--- LAKE CREEK.prj (project) ---

Proj Title=LAKE CREEK Base Level Engineering
Current Plan=p01
Default Exp/Contr=0.3,0.1
English Units
Geom File=g01
Flow File=f01
Flow File=f02
Plan File=p01
Y Axis Title=Elevation
X Axis Title(PF)=Main Channel Distance
X Axis Title(XS)=Station
BEGIN DESCRIPTION:
LAKE CREEK
END DESCRIPTION:
DSS Export Rating Curves= 0
DSS Export Rating Curve Sorted= 0
DSS Export Volume Flow Curves= 0
DXF OffsetX= 0
DXF OffsetY= 0
DXF ScaleX= 1
DXF ScaleY= 10

--- LAKE CREEK.p01 (plan) ---

Plan Title=Multiple Run
Short Identifier=Multiple
Geom File=g01
Flow File=f01
Subcritical Flow
K Sum by GR= 0
Std Step Tol= 0.01
Critical Tol= 0.01
Num of Std Step Trials= 20
Max Error Tol= 0.3
Flow Tol Ratio= 0.001
Split Flow NTrial= 30
Split Flow Tol= 0.02
Split Flow Ratio= 0.02
Log Output Level= 0
Friction Slope Method= 1
Unsteady Friction Slope Method= 2
Unsteady Bridges Friction Slope Method= 1
Parabolic Critical Depth
Global Vel Dist=  1 , 1 , 1
Global Log Level= 0
CheckData=True
Encroach Param= -1, 0, 0, 0
BEGIN DESCRIPTION:
Multiple Run
END DESCRIPTION:

--- LAKE CREEK.f01 (steady flow) ---

Flow Title=Multiple
Program Version=4.10
Number of Profiles= 7
Profile Names=10-year,25-year,50-year,1pct_min,100-year,1pct_plu,500-year
River Rch & RM=LAKE CREEK,Reach-1         ,358856
     639     869    1176     524    1583    4781    2964
River Rch & RM=LAKE CREEK,Reach-1         ,349809
    1404    1985    2759    1257    3797   11467    7449
River Rch & RM=LAKE CREEK,Reach-1         ,342475
    3190    4649    6596    3061    9244   27916   18808
River Rch & RM=LAKE CREEK,Reach-1         ,336405
    3322    4843    6872    3188    9629   29079   19582
River Rch & RM=LAKE CREEK,Reach-1         ,334000
    3321    4837    6861    3181    9607   29013   19517
River Rch & RM=LAKE CREEK,Reach-1         ,333000
    3542    5166    7332    3402   10275   31030   20896
River Rch & RM=LAKE CREEK,Reach-1         ,331000
    3703    5402    7667    3557   10741   32437   21835
River Rch & RM=LAKE CREEK,Reach-1         ,328500
    3785    5499    7784    3600   10871   32830   21959
River Rch & RM=LAKE CREEK,Reach-1         ,322500
    3915    5695    8067    3734   11275   34050   22811
River Rch & RM=LAKE CREEK,Reach-1         ,322000
    4517    6589    9354    4336   13094   39543   26574
River Rch & RM=LAKE CREEK,Reach-1         ,314500
    4827    7040    9991    4629   13979   42216   28339
River Rch & RM=LAKE CREEK,Reach-1         ,308375
    6424    9448   13490    6283   18975   57304   38872
River Rch & RM=LAKE CREEK,Reach-1         ,307830
    6750    9927   14170    6599   19928   60182   40800
River Rch & RM=LAKE CREEK,Reach-1         ,306500
    6750    9927   14170    6599   19928   60182   40800
River Rch & RM=LAKE CREEK,Reach-1         ,300318
    6798    9993   14260    6638   20046   60538   41010
River Rch & RM=LAKE CREEK,Reach-1         ,298000
    6737    9889   14098    6556   19798   59789   40417
River Rch & RM=LAKE CREEK,Reach-1         ,295338
    7105   10443   14902    6935   20944   63250   42828
River Rch & RM=LAKE CREEK,Reach-1         ,292500
    7193   10572   15087    7021   21203   64032   43356
River Rch & RM=LAKE CREEK,Reach-1         ,290894
    7170   10525   15005    6977   21069   63627   42998
River Rch & RM=LAKE CREEK,Reach-1         ,287118
    7119   10409   14799    6861   20721   62576   42039
River Rch & RM=LAKE CREEK,Reach-1         ,286460
    7119   10409   14799    6861   20721   62576   42039
River Rch & RM=LAKE CREEK,Reach-1         ,276500
    7056   10307   14644    6784   20488   61873   41507
River Rch & RM=LAKE CREEK,Reach-1         ,274498
    7412   10833   15400    7137   21554   65092   43698
River Rch & RM=LAKE CREEK,Reach-1         ,272139
    7605   11128   15832    7343   22175   66967   45024
River Rch & RM=LAKE CREEK,Reach-1         ,270440
    7700   11272   16041    7442   22474   67870   45661
River Rch & RM=LAKE CREEK,Reach-1         ,267720
   10561   15566   22263   10375   31333   94624   64208
River Rch & RM=LAKE CREEK,Reach-1         ,260966
   10655   15668   22371   10408   31431   94920   64180
River Rch & RM=LAKE CREEK,Reach-1         ,252000
   10655   15668   22371   10408   31431   94920   64180
River Rch & RM=LAKE CREEK,Reach-1         ,248000
   10746   15798   22554   10492   31684   95684   64674
River Rch & RM=LAKE CREEK,Reach-1         ,246759
   11166   16407   23414   10887   32877   99287   67046
River Rch & RM=LAKE CREEK,Reach-1         ,240000
   10992   16117   22969   10664   32204   97255   65475
River Rch & RM=LAKE CREEK,Reach-1         ,227021
   11486   16812   23933   11099   33519  101226   67976
River Rch & RM=LAKE CREEK,Reach-1         ,219793
   11415   16731   23840   11064   33414  100909   67894
River Rch & RM=LAKE CREEK,Reach-1         ,219000
   11620   16992   24175   11204   33836  102183   68528
River Rch & RM=LAKE CREEK,Reach-1         ,213829
   11619   16947   24071   11135   33628  101555   67857
River Rch & RM=LAKE CREEK,Reach-1         ,201940
   11769   17153   24351   11258   34000  102678   68525
River Rch & RM=LAKE CREEK,Reach-1         ,191914
   11843   17262   24507   11331   34220  103343   68977
River Rch & RM=LAKE CREEK,Reach-1         ,189735
   14194   20732   29480   13651   41224  124494   83306
River Rch & RM=LAKE CREEK,Reach-1         ,182928
   14196   20735   29484   13652   41228  124507   83313
River Rch & RM=LAKE CREEK,Reach-1         ,181530
   14328   20926   29759   13779   41613  125669   84091
River Rch & RM=LAKE CREEK,Reach-1         ,176927
   14288   20861   29657   13729   41462  125213   83740
River Rch & RM=LAKE CREEK,Reach-1         ,175805
   14287   20857   29648   13723   41444  125159   83688
River Rch & RM=LAKE CREEK,Reach-1         ,174899
   14194   20703   29412   13606   41088  124084   82866
River Rch & RM=LAKE CREEK,Reach-1         ,168971
   14126   20587   29232   13514   40812  123250   82216
River Rch & RM=LAKE CREEK,Reach-1         ,165824
   17558   25681   36567   16951   51190  154591  103630
River Rch & RM=LAKE CREEK,Reach-1         ,163000
   17776   26005   37032   17169   51849  156581  104989
River Rch & RM=LAKE CREEK,Reach-1         ,156351
   17825   26073   37127   17211   51977  156968  105231
River Rch & RM=LAKE CREEK,Reach-1         ,152177
   17724   25905   36868   17082   51587  155790  104327
River Rch & RM=LAKE CREEK,Reach-1         ,147837
   18405   26858   38190   17679   53391  161238  107748
River Rch & RM=LAKE CREEK,Reach-1         ,144904
   18922   27607   39252   18168   54865  165690  110685
River Rch & RM=LAKE CREEK,Reach-1         ,139839
   19128   27902   39667   18358   55440  167426  111817
River Rch & RM=LAKE CREEK,Reach-1         ,134000
   19125   27873   39599   18315   55310  167034  111404
River Rch & RM=LAKE CREEK,Reach-1         ,126188
   19125   27873   39599   18315   55310  167034  111404
River Rch & RM=LAKE CREEK,Reach-1         ,125000
   19146   27886   39603   18309   55292  166979  111272
River Rch & RM=LAKE CREEK,Reach-1         ,123847
   19193   27948   39685   18344   55397  167296  111446
River Rch & RM=LAKE CREEK,Reach-1         ,119032
   19193   27948   39685   18344   55397  167296  111446
River Rch & RM=LAKE CREEK,Reach-1         ,117000
   19257   28009   39743   18355   55432  167402  111336
River Rch & RM=LAKE CREEK,Reach-1         ,109357
   19257   28009   39743   18355   55432  167402  111336
River Rch & RM=LAKE CREEK,Reach-1         ,103711
   19101   27742   39323   18143   54790  165463  109813
River Rch & RM=LAKE CREEK,Reach-1         ,90132
   19248   27950   39613   18274   55188  166665  110581
River Rch & RM=LAKE CREEK,Reach-1         ,87000
   19549   28385   40228   18557   56042  169244  112278
River Rch & RM=LAKE CREEK,Reach-1         ,82773
   19480   28271   40056   18472   55784  168465  111692
River Rch & RM=LAKE CREEK,Reach-1         ,81000
   19585   28395   40203   18526   55948  168960  111853
River Rch & RM=LAKE CREEK,Reach-1         ,66728
   19585   28395   40203   18526   55948  168960  111853
River Rch & RM=LAKE CREEK,Reach-1         ,64363
   20343   29454   41671   19188   57948  175000  115639
River Rch & RM=LAKE CREEK,Reach-1         ,53000
   20343   29454   41671   19188   57948  175000  115639
River Rch & RM=LAKE CREEK,Reach-1         ,50000
   20416   29556   41812   19252   58140  175580  116004
River Rch & RM=LAKE CREEK,Reach-1         ,45042
   20415   29551   41803   19246   58123  175529  115957
River Rch & RM=LAKE CREEK,Reach-1         ,44395
   20460   29613   41888   19284   58236  175870  116160
River Rch & RM=LAKE CREEK,Reach-1         ,40899
   20460   29613   41888   19284   58236  175870  116160
River Rch & RM=LAKE CREEK,Reach-1         ,40632
   21439   31038   43914   20222   61068  184422  121855
River Rch & RM=LAKE CREEK,Reach-1         ,39384
   21439   31038   43914   20222   61068  184422  121855
River Rch & RM=LAKE CREEK,Reach-1         ,31779
   21462   31068   43955   20239   61121  184582  121946
River Rch & RM=LAKE CREEK,Reach-1         ,29940
   21741   31463   44504   20488   61872  186850  123391
River Rch & RM=LAKE CREEK,Reach-1         ,25000
   21741   31463   44504   20488   61872  186850  123391
River Rch & RM=LAKE CREEK,Reach-1         ,22191
   21750   31465   44497   20480   61848  186778  123279
River Rch & RM=LAKE CREEK,Reach-1         ,17000
   21670   31333   44296   20379   61545  185863  122588
River Rch & RM=LAKE CREEK,Reach-1         ,11221
   21550   31132   43984   20224   61074  184441  121494
River Rch & RM=LAKE CREEK,Reach-1         ,3866
   21529   31088   43907   20182   60948  184060  121165
Boundary for River Rch & Prof#=LAKE CREEK,Reach-1         , 1
Up Type= 0
Dn Type= 3
Dn Slope=0.0005
Boundary for River Rch & Prof#=LAKE CREEK,Reach-1         , 2
Up Type= 0
Dn Type= 3
Dn Slope=0.0005
Boundary for River Rch & Prof#=LAKE CREEK,Reach-1         , 3
Up Type= 0
Dn Type= 3
Dn Slope=0.0005
Boundary for River Rch & Prof#=LAKE CREEK,Reach-1         , 4
Up Type= 0
Dn Type= 3
Dn Slope=0.0005
Boundary for River Rch & Prof#=LAKE CREEK,Reach-1         , 5
Up Type= 0
Dn Type= 3
Dn Slope=0.0005
Boundary for River Rch & Prof#=LAKE CREEK,Reach-1         , 6
Up Type= 0
Dn Type= 3
Dn Slope=0.0005
Boundary for River Rch & Prof#=LAKE CREEK,Reach-1         , 7
Up Type= 0
Dn Type= 3
Dn Slope=0.0005
DSS Import GetInterval= 0
DSS Import GetPeak= 0
DSS Import FillOption= 0

--- LAKE CREEK.f02 (steady flow) ---

Flow Title=Orig_BLE_Flows
Program Version=4.10
Number of Profiles= 7
Profile Names=10-year,25-year,50-year,1pct_min,100-year,1pct_plu,500-year
River Rch & RM=LAKE CREEK,Reach-1         ,358856
     639     852    1023     403    1218    3678    1723
River Rch & RM=LAKE CREEK,Reach-1         ,349809
    1404    1946    2399     967    2921    8820    4331
River Rch & RM=LAKE CREEK,Reach-1         ,342475
    3190    4558    5736    2355    7111   21476   10935
River Rch & RM=LAKE CREEK,Reach-1         ,336405
    3322    4748    5976    2453    7407   22368   11385
River Rch & RM=LAKE CREEK,Reach-1         ,334000
    3321    4742    5966    2447    7390   22318   11347
River Rch & RM=LAKE CREEK,Reach-1         ,333000
    3542    5065    6376    2617    7904   23868   12149
River Rch & RM=LAKE CREEK,Reach-1         ,331000
    3703    5296    6667    2736    8262   24952   12695
River Rch & RM=LAKE CREEK,Reach-1         ,328500
    3785    5391    6769    2769    8362   25253   12767
River Rch & RM=LAKE CREEK,Reach-1         ,322500
    3915    5583    7015    2872    8673   26191   13262
River Rch & RM=LAKE CREEK,Reach-1         ,322000
    4517    6460    8134    3335   10072   30418   15450
River Rch & RM=LAKE CREEK,Reach-1         ,314500
    4827    6902    8688    3561   10753   32474   16476
River Rch & RM=LAKE CREEK,Reach-1         ,308375
    6424    9263   11730    4833   14596   44079   22600
River Rch & RM=LAKE CREEK,Reach-1         ,307830
    6750    9732   12322    5076   15329   46293   23721
River Rch & RM=LAKE CREEK,Reach-1         ,306500
    6750    9732   12322    5076   15329   46293   23721
River Rch & RM=LAKE CREEK,Reach-1         ,300318
    6798    9797   12400    5106   15420   46568   23843
River Rch & RM=LAKE CREEK,Reach-1         ,298000
    6737    9695   12259    5043   15229   45990   23498
River Rch & RM=LAKE CREEK,Reach-1         ,295338
    7105   10238   12958    5335   16111   48655   24900
River Rch & RM=LAKE CREEK,Reach-1         ,292500
    7193   10365   13119    5401   16310   49257   25207
River Rch & RM=LAKE CREEK,Reach-1         ,290894
    7170   10319   13048    5367   16207   48945   24999
River Rch & RM=LAKE CREEK,Reach-1         ,287115
    7119   10205   12869    5278   15939   48134   24441
River Rch & RM=LAKE CREEK,Reach-1         ,286460
    7119   10205   12869    5278   15939   48134   24441
River Rch & RM=LAKE CREEK,Reach-1         ,276500
    7056   10105   12734    5219   15760   47595   24132
River Rch & RM=LAKE CREEK,Reach-1         ,274498
    7412   10621   13391    5490   16580   50070   25406
River Rch & RM=LAKE CREEK,Reach-1         ,272139
    7605   10910   13767    5648   17058   51513   26177
River Rch & RM=LAKE CREEK,Reach-1         ,270440
    7700   11051   13949    5725   17288   52210   26547
River Rch & RM=LAKE CREEK,Reach-1         ,267720
   10561   15261   19359    7981   24102   72788   37330
River Rch & RM=LAKE CREEK,Reach-1         ,260966
   10655   15361   19453    8006   24178   73016   37314
River Rch & RM=LAKE CREEK,Reach-1         ,252000
   10655   15361   19453    8006   24178   73016   37314
River Rch & RM=LAKE CREEK,Reach-1         ,248000
   10746   15488   19612    8070   24372   73601   37601
River Rch & RM=LAKE CREEK,Reach-1         ,246759
   11166   16085   20360    8374   25290   76375   38980
River Rch & RM=LAKE CREEK,Reach-1         ,240000
   10992   15801   19973    8203   24772   74810   38067
River Rch & RM=LAKE CREEK,Reach-1         ,227021
   11486   16482   20811    8538   25784   77866   39521
River Rch & RM=LAKE CREEK,Reach-1         ,219793
   11415   16403   20730    8511   25703   77623   39473
River Rch & RM=LAKE CREEK,Reach-1         ,219000
   11620   16659   21022    8619   26028   78604   39842
River Rch & RM=LAKE CREEK,Reach-1         ,213829
   11619   16615   20931    8566   25868   78121   39452
River Rch & RM=LAKE CREEK,Reach-1         ,201940
   11769   16817   21175    8660   26154   78984   39840
River Rch & RM=LAKE CREEK,Reach-1         ,191914
   11843   16924   21310    8717   26323   79496   40103
River Rch & RM=LAKE CREEK,Reach-1         ,189735
   14194   20325   25635   10500   31711   95766   48434
River Rch & RM=LAKE CREEK,Reach-1         ,182928
   14196   20328   25638   10502   31714   95776   48438
River Rch & RM=LAKE CREEK,Reach-1         ,181530
   14328   20516   25877   10599   32010   96668   48890
River Rch & RM=LAKE CREEK,Reach-1         ,176927
   14288   20452   25789   10561   31894   96317   48686
River Rch & RM=LAKE CREEK,Reach-1         ,175805
   14287   20448   25781   10557   31880   96277   48656
River Rch & RM=LAKE CREEK,Reach-1         ,174899
   14194   20297   25576   10466   31606   95450   48178
River Rch & RM=LAKE CREEK,Reach-1         ,168971
   14126   20183   25419   10396   31394   94809   47800
River Rch & RM=LAKE CREEK,Reach-1         ,165824
   17558   25177   31797   13039   39377  118916   60250
River Rch & RM=LAKE CREEK,Reach-1         ,163000
   17776   25495   32202   13207   39884  120446   61040
River Rch & RM=LAKE CREEK,Reach-1         ,156351
   17825   25562   32284   13239   39982  120745   61181
River Rch & RM=LAKE CREEK,Reach-1         ,152177
   17724   25397   32059   13140   39682  119838   60655
River Rch & RM=LAKE CREEK,Reach-1         ,147837
   18405   26331   33209   13599   41070  124028   62644
River Rch & RM=LAKE CREEK,Reach-1         ,144904
   18922   27066   34132   13975   42204  127455   64352
River Rch & RM=LAKE CREEK,Reach-1         ,139839
   19128   27355   34493   14122   42646  128790   65010
River Rch & RM=LAKE CREEK,Reach-1         ,134000
   19125   27326   34434   14088   42546  128486   64770
River Rch & RM=LAKE CREEK,Reach-1         ,126188
   19125   27326   34434   14088   42546  128486   64770
River Rch & RM=LAKE CREEK,Reach-1         ,125000
   19146   27339   34437   14084   42532  128444   64693
River Rch & RM=LAKE CREEK,Reach-1         ,123847
   19193   27400   34509   14110   42613  128689   64794
River Rch & RM=LAKE CREEK,Reach-1         ,119032
   19193   27400   34509   14110   42613  128689   64794
River Rch & RM=LAKE CREEK,Reach-1         ,117000
   19257   27460   34559   14120   42640  128771   64730
River Rch & RM=LAKE CREEK,Reach-1         ,109357
   19257   27460   34559   14120   42640  128771   64730
River Rch & RM=LAKE CREEK,Reach-1         ,103711
   19101   27198   34194   13956   42146  127279   63845
River Rch & RM=LAKE CREEK,Reach-1         ,90132
   19248   27402   34446   14057   42452  128202   64291
River Rch & RM=LAKE CREEK,Reach-1         ,87000
   19549   27828   34981   14275   43109  130186   65278
River Rch & RM=LAKE CREEK,Reach-1         ,82773
   19480   27717   34831   14209   42911  129589   64937
River Rch & RM=LAKE CREEK,Reach-1         ,81000
   19585   27838   34959   14251   43037  129969   65031
River Rch & RM=LAKE CREEK,Reach-1         ,66728
   19585   27838   34959   14251   43037  129969   65031
River Rch & RM=LAKE CREEK,Reach-1         ,64363
   20343   28876   36236   14760   44575  134615   67232
River Rch & RM=LAKE CREEK,Reach-1         ,53000
   20343   28876   36236   14760   44575  134615   67232
River Rch & RM=LAKE CREEK,Reach-1         ,50000
   20416   28976   36358   14809   44723  135060   67444
River Rch & RM=LAKE CREEK,Reach-1         ,45042
   20415   28972   36350   14805   44710  135023   67417
River Rch & RM=LAKE CREEK,Reach-1         ,44395
   20460   29032   36424   14834   44797  135283   67535
River Rch & RM=LAKE CREEK,Reach-1         ,40899
   20460   29032   36424   14834   44797  135283   67535
River Rch & RM=LAKE CREEK,Reach-1         ,40632
   21439   30429   38186   15555   46975  141863   70846
River Rch & RM=LAKE CREEK,Reach-1         ,39384
   21439   30429   38186   15555   46975  141863   70846
River Rch & RM=LAKE CREEK,Reach-1         ,31779
   21462   30459   38222   15569   47016  141987   70899
River Rch & RM=LAKE CREEK,Reach-1         ,29940
   21741   30846   38699   15760   47594  143732   71739
River Rch & RM=LAKE CREEK,Reach-1         ,25000
   21741   30846   38699   15760   47594  143732   71739
River Rch & RM=LAKE CREEK,Reach-1         ,22191
   21750   30848   38693   15753   47575  143674   71674
River Rch & RM=LAKE CREEK,Reach-1         ,17000
   21670   30719   38518   15676   47342  142971   71272
River Rch & RM=LAKE CREEK,Reach-1         ,11221
   21550   30522   38247   15557   46980  141877   70636
River Rch & RM=LAKE CREEK,Reach-1         ,3866
   21529   30478   38180   15524   46883  141583   70445
Boundary for River Rch & Prof#=LAKE CREEK,Reach-1         , 1
Up Type= 0
Dn Type= 3
Dn Slope=0.0005
Boundary for River Rch & Prof#=LAKE CREEK,Reach-1         , 2
Up Type= 0
Dn Type= 3
Dn Slope=0.0005
Boundary for River Rch & Prof#=LAKE CREEK,Reach-1         , 3
Up Type= 0
Dn Type= 3
Dn Slope=0.0005
Boundary for River Rch & Prof#=LAKE CREEK,Reach-1         , 4
Up Type= 0
Dn Type= 3
Dn Slope=0.0005
Boundary for River Rch & Prof#=LAKE CREEK,Reach-1         , 5
Up Type= 0
Dn Type= 3
Dn Slope=0.0005
Boundary for River Rch & Prof#=LAKE CREEK,Reach-1         , 6
Up Type= 0
Dn Type= 3
Dn Slope=0.0005
Boundary for River Rch & Prof#=LAKE CREEK,Reach-1         , 7
Up Type= 0
Dn Type= 3
Dn Slope=0.0005
DSS Import GetInterval= 0
DSS Import GetPeak= 0
DSS Import FillOption= 0

--- LAKE CREEK.g01 (geometry) ---

Geom Title=Existing Conditions
Program Version=4.10

River Reach=LAKE CREEK      ,Reach-1
Reach XY= 30
      3690584.38     10222801.59      3692215.46      10217129.7
      3698706.25     10217008.99       3702500.8     10208246.17
      3707184.65     10203539.24      3706930.37     10197445.15
      3714021.03     10185262.72      3718902.56     10181030.29
      3719371.12     10173985.28       3728011.5       10167657.
      3728229.74     10157608.32      3732831.05     10148505.59
      3734930.01     10148349.99      3735379.17     10128771.13
       3737374.7     10123280.59      3743325.91      10118726.8
      3742361.33     10112755.24      3746623.82     10109630.83
      3749161.15     10103294.08      3754711.27     10102094.21
      3757258.71     10095706.23      3762888.15     10093987.06
      3767166.59     10085878.11      3784671.28     10082647.16
      3788231.57      10085055.7      3791868.32     10084308.87
        3798817.     10089266.23      3808043.71     10090049.96
      3816081.63     10096535.64      3824049.75     10094306.84

Type RM Length L Ch R = 1 ,358856  ,356,356,356
BEGIN DESCRIPTION:
LAKE CREEK 696.0
END DESCRIPTION:
XS GIS Cut Line= 3
      3691165.31     10222932.96      3690628.89     10222656.94
      3690035.18     10222573.61
#Sta/Elev= 30
  4404.7  386.07  4435.6  384.76    4447  385.37    4458  384.36  4491.8  384.81
  4507.9  383.88  4581.8  383.68    4624  381.91    4641  382.15  4657.5   381.1
  4694.2  381.45  4729.7  379.71  4751.8  380.18  4790.6  378.93  4834.9  379.93
  4873.6  378.96  4879.3  380.02  4907.9  378.23  4926.7  378.05  4952.9  377.03
  4968.7  377.44  4990.1   376.9    5011   376.2  5012.4   375.5  5029.2  377.23
  5150.4  379.02  5180.7  380.45  5241.3   381.5    5442  380.66  5607.5  384.34
#Mann= 6 ,-1 , 0
  4404.7     .17       0    4624     .11       0  4926.7     .15       0
  4968.7     .11       0  4990.1     .06       0  5029.2     .11       0
Bank Sta=4990.1,5029.2
XS Rating Curve= 0 ,0
Exp/Cntr=0.3,0.1

Type RM Length L Ch R = 1 ,358500  ,454,454,454
BEGIN DESCRIPTION:
LAKE CREEK 695.0
END DESCRIPTION:
XS GIS Cut Line= 3
      3691467.88     10222811.09      3690675.06     10222312.43
      3690010.95     10222365.12
#Sta/Elev= 30
  4063.4  390.02  4098.9  389.88  4144.1   388.1  4238.3  387.36  4274.8  385.49
  4374.9  383.87  4390.2  382.98  4453.8  383.01    4536  380.73  4636.3  380.26
  4651.6   379.3  4694.1  378.66  4715.3     379  4730.6   378.2  4918.9  376.19
  4955.5  375.38  4976.7  375.85  4994.8  373.64  5027.3  376.07  5117.6  378.08
  5148.8  377.74  5187.8  379.07  5197.8  378.64  5207.9  379.58    5258  380.12
  5358.3  379.98  5398.5  378.65  5424.4  378.78  5649.2  384.43  5666.2  386.01
#Mann= 5 ,-1 , 0
  4063.4     .11       0  4918.9     .15       0  4976.7     .06       0
  5027.3     .15       0  5148.8     .11       0
Bank Sta=4976.7,5027.3
XS Rating Curve= 0 ,0
Exp/Cntr=0.3,0.1

Type RM Length L Ch R = 1 ,358046  ,497,497,497
BEGIN DESCRIPTION:
LAKE CREEK 694.0
END DESCRIPTION:
XS GIS Cut Line= 3
      3691267.84     10222211.06      3690597.64     10221839.23
      3689967.89     10222261.04
#Sta/Elev= 30
  4132.3   382.3  4227.3  381.47  4302.8  378.96  4514.5  377.01  4714.8  373.65
  4913.8   371.9  4949.8  373.08  4970.8  372.02  4984.1  370.63  4994.8  371.46
  5030.8  371.51  5036.9  372.44  5042.9  372.01  5066.9  373.44  5078.8     373
  5115.1  372.52  5138.9   374.1  5144.9  373.15  5174.9  373.15    5232  375.37
    5247  374.79  5259.6  375.86    5325  375.98  5397.1  377.43  5440.1  379.49
  5463.1  379.23  5535.2  381.15  5613.2  383.96  5628.2  385.27  5656.7  385.81
#Mann= 4 ,-1 , 0
  4132.3     .11       0  4970.8     .06       0  5036.9     .15       0
  5078.8     .11       0
Bank Sta=4970.8,5036.9
XS Rating Curve= 0 ,0
Exp/Cntr=0.3,0.1

Type RM Length L Ch R = 1 ,357549  ,549,549,549
BEGIN DESCRIPTION:
LAKE CREEK 693.0
END DESCRIPTION:
XS GIS Cut Line= 4
      3690957.01     10221912.15      3690462.22     10221594.44
      3690134.84     10221403.87      3689946.66     10221637.17
#Sta/Elev= 30
       0  376.24   101.9  373.83   310.7  372.26     341   370.6   362.2  370.91
   404.5  370.43   419.7  369.67   471.2  369.99   498.3  369.39   507.5   369.9
   528.7  369.48   543.9  369.85   549.8  370.59     565  368.94   570.9  369.32
   586.1  368.54   623.3  368.34   650.9  369.46   870.8  370.14   901.3  371.03
   944.3  370.96   964.6  372.24   990.6  370.85  1019.4  370.83  1062.6  372.25
  1118.6  372.17  1147.4   374.4  1176.1  373.34  1219.3  373.96  1265.8  375.85
#Mann= 3 , 0 , 0
       0     .11       0   570.9     .06       0   650.9     .11       0
Bank Sta=570.9,650.9
XS Rating Curve= 0 ,0
Exp/Cntr=0.3,0.1

Type RM Length L Ch R = 1 ,357000  ,500,500,500
BEGIN DESCRIPTION:
LAKE CREEK 692.0
END DESCRIPTION:
XS GIS Cut Line= 3
      3691217.85     10221611.07      3690827.08     10221198.29
      3690337.21     10221037.14
#Sta/Elev= 30
  4431.6  376.27  4558.8  374.05  4665.2  371.32  4672.1   371.6  4679.4  370.74
  4686.2  371.03  4714.6  369.79  4735.6  369.94  4742.9  369.22  4763.9  369.23
  4785.3  368.22  4834.7  368.09  4848.9  367.08  4870.3  367.62  4941.1  365.18
    4958  365.38  4976.3  365.37  5002.2  364.04    5004  363.24  5007.5  363.24
    5011  364.48  5020.2  365.67  5051.8  364.64  5101.2  366.01  5138.2  367.87
  5233.6  368.54  5260.1  369.78  5283.4  369.47  5450.9  371.53  5515.7  371.09
#Mann= 4 ,-1 , 0
  4431.6     .11       0    4958     .17       0  4976.3     .06       0
  5020.2     .11       0
Bank Sta=4976.3,5020.2
XS Rating Curve= 0 ,0
Exp/Cntr=0.3,0.1

Type RM Length L Ch R = 1 ,356500  ,530,530,530
BEGIN DESCRIPTION:
LAKE CREEK 691.0
END DESCRIPTION:
XS GIS Cut Line= 3
      3691524.69     10221089.21      3690994.16     10220801.34
      3690457.02     10220854.85
#Sta/Elev= 30
  4396.4  368.87  4415.6     369  4575.6  366.15  4586.1  366.34  4597.6   365.7
  4629.8  365.53  4657.4  364.65  4673.6  364.85  4717.3  364.09    4723  363.46
  4813.8   362.6  4820.9  363.08  4842.8  363.15  4859.2  361.85  4893.4  360.81
  4916.2  362.02  4930.2  361.12  4952.1  360.35  4984.4  360.54  4993.1  360.27
  4993.3  359.77  5026.4  361.36  5056.6  361.59    5137  364.21  5227.4  365.44
  5257.6  366.82  5317.9  366.75  5368.1  368.25  5408.3   368.2  5539.8  369.81
#Mann= 4 ,-1 , 0
  4396.4     .11       0  4859.2     .17       0  4930.2     .06       0
  5026.4     .11       0
Bank Sta=4930.2,5026.4
XS Rating Curve= 0 ,0
Exp/Cntr=0.3,0.1

Type RM Length L Ch R = 1 ,355970  ,470,470,470
BEGIN DESCRIPTION:
LAKE CREEK 690.0
END DESCRIPTION:
XS GIS Cut Line= 3
      3691441.44      10220443.4      3690967.43     10220354.85
      3690545.59     10220620.46
#Sta/Elev= 30
  4502.7  359.56  4658.9  358.49    4742   357.1  4763.1  356.14    4781  356.74
  4801.4  356.33  4868.4  356.95  4926.4  358.47  4964.1  357.66  4973.7  357.95
  4978.8  357.49  4982.1  355.74  4984.9  355.74  4988.8  357.19  4994.5  354.41
    4998  354.41  4998.2  354.91    5004  356.01  5031.7  356.42  5040.5  356.05
  5061.7  356.86  5155.9  358.71  5207.7  360.35  5359.6  363.19  5386.7  365.26
  5409.8  365.52  5417.3   365.1  5423.2  365.82  5453.8  365.01  5483.4  365.94
#Mann= 5 ,-1 , 0
  4502.7     .11       0    4742     .17       0  4926.4     .11       0
  4988.8     .06       0  5061.7     .11       0
Bank Sta=4988.8,5061.7
XS Rating Curve= 0 ,0
Exp/Cntr=0.3,0.1

Type RM Length L Ch R = 1 ,355500  ,728,728,728
BEGIN DESCRIPTION:
LAKE CREEK 689.0
END DESCRIPTION:
XS GIS Cut Line= 4
      3691441.38     10220261.09      3690980.76     10219903.06
      3690811.04     10219887.65      3690608.05     10220235.07
#Sta/Elev= 30
  4416.6  357.31  4525.6  355.75    4598  355.69  4703.9  353.58  4867.7  352.36
  4889.7  351.72  4911.2  352.73  4917.5   352.3  4946.4  352.46  4960.9  351.33
  4981.7  350.59  4989.9  348.61  4996.2  349.68  4996.9  347.53    5004  348.03
    5023  351.41    5033  350.72  5072.7  350.89  5083.3  351.58  5113.4  350.76
  5189.2  351.97  5255.5  351.95  5269.4  352.54  5322.3  352.67  5417.6  354.42
  5439.7  354.24  5482.6  355.39  5541.3  356.06  5562.8  356.93  5572.8  356.71
#Mann= 3 , 0 , 0
  4416.6     .11       0  4981.7     .06       0    5023     .11       0
Bank Sta=4981.7,5023
XS Rating Curve= 0 ,0
Exp/Cntr=0.3,0.1

Type RM Length L Ch R = 1 ,354772  ,636,636,636
BEGIN DESCRIPTION:
LAKE CREEK 688.0
END DESCRIPTION:
XS GIS Cut Line= 3
      3691524.74      10220302.8      3691003.89     10219584.02
      3690404.98     10219292.38
#Sta/Elev= 30
  4098.1  357.75  4124.9  356.67  4183.5  356.88  4325.8  355.48    4506  352.52
  4577.1  352.93  4662.9  351.16  4698.5  351.48  4727.9  350.62  4769.6  351.07
    4799  350.08  4819.9  350.63  4849.3  349.37  4964.5  347.48    4977  347.04
  4984.5  345.45    4999  343.43  4999.2  342.93  5002.7  342.93  5006.5  344.58
  5014.7  345.77  5068.6  346.72  5096.7  346.03  5148.2  346.12  5254.5  347.53
  5282.6   347.3  5299.6  348.24  5337.3  348.36  5367.2  349.62  5651.9  356.37
#Mann= 3 , 0 , 0
  4098.1     .11       0  4984.5     .06       0  5014.7     .11       0
Bank Sta=4984.5,5014.7
XS Rating Curve= 0 ,0
Exp/Cntr=0.3,0.1

Type RM Length L Ch R = 1 ,354136  ,614,614,614
BEGIN DESCRIPTION:
LAKE CREEK 686.0
END DESCRIPTION:
XS GIS Cut Line= 3
      3691717.86     10219461.08      3691253.89     10219172.56
      3690425.78     10218979.86
#Sta/Elev= 30
    4446  353.12  4575.5  350.37  4634.4  350.01  4657.9  349.19  4663.8  349.68
  4693.3  348.07  4706.3  348.18  4728.6  347.15  4800.8  347.23  4810.2  345.84
  4953.1  342.96  4975.9  342.13  4996.6  340.01  4996.8  339.51  5008.8   340.6
  5022.6  343.04  5029.4  343.63    5091  342.89  5101.2  343.46  5224.4  342.86
  5316.8  343.75  5421.4  346.23    5464  346.65  5470.9  347.28  5639.5  351.05
  5676.2  352.61  5729.8  353.89  5748.1  353.83    5815  355.69  5842.6  355.56
#Mann= 3 ,-1 , 0
    4446     .11       0  4953.1     .06       0  5022.6     .11       0
Bank Sta=4953.1,5022.6
XS Rating Curve= 0 ,0
Exp/Cntr=0.3,0.1

Type RM Length L Ch R = 1 ,353522  ,398,398,398
BEGIN DESCRIPTION:
LAKE CREEK 685.0
END DESCRIPTION:
XS GIS Cut Line= 3
      3691917.88     10219011.09      3691436.18     10218750.69
      3690555.94      10218880.9
#Sta/Elev= 30
    4525  353.57  4576.9   351.5  4604.6  349.42  4672.8  347.03  4730.1  346.32
  4768.2  344.99  4775.1  344.16  4828.1  342.53  4866.1  342.18  4900.2  340.55
  4981.3  339.97  4991.1  339.02  4995.7  336.42  4999.2  336.42  5003.2  338.28
  5013.7  340.49    5081  339.91  5131.5   341.2  5222.5  341.08  5495.5  349.98
  5535.9  350.27  5606.7  348.54  5659.2  348.16  5677.4  348.86  5697.6   348.7
  5728.7  349.98  5778.5  348.89  5798.7  349.48  5829.1  349.28  5962.4  352.11
#Mann= 3 , 0 , 0
    4525     .11       0  4981.3     .06       0  5013.7     .11       0
Bank Sta=4981.3,5013.7
XS Rating Curve= 0 ,0
Exp/Cntr=0.3,0.1

Type RM Length L Ch R = 1 ,353124  ,624,624,624
BEGIN DESCRIPTION:
LAKE CREEK 684.0
END DESCRIPTION:
XS GIS Cut Line= 3
      3692009.09      10218761.1      3691712.22     10218474.65
      3690998.72     10218729.84
#Sta/Elev= 30
  4598.3  350.69  4620.4   351.4  4655.7  350.66  4740.5  347.13  4768.8  345.12
  4802.7   344.3  4875.1  341.93  4938.6  340.96  4974.1  338.81  4988.3  337.26
  4993.2  336.49  4993.5  335.99    4997  335.99  4997.2  336.49  5002.4   337.7
  5009.4  337.31  5017.9  338.78  5068.6  338.61  5079.5  339.15  5130.4  337.99
  5197.3  338.67  5206.6  338.13  5284.3  339.71  5309.8   338.7  5402.1  339.24
  5576.2  343.61  5631.5  345.99  5668.5  346.49  5673.9  347.43  5768.6  349.67
#Mann= 4 ,-1 , 0
  4598.3     .17       0  4802.7     .11       0  4974.1     .06       0
  5017.9     .11       0
Bank Sta=4974.1,5017.9
XS Rating Curve= 0 ,0
Exp/Cntr=0.3,0.1

Type RM Length L Ch R = 1 ,352500  ,500,500,500
BEGIN DESCRIPTION:
LAKE CREEK 683.0
END DESCRIPTION:
XS GIS Cut Line= 3
      3692117.83     10218561.05      3691608.67      10217927.1
      3691267.81     10217861.06
#Sta/Elev= 30
  4186.9  346.32  4214.9  346.39  4222.9  345.43  4229.3  345.92  4282.8   345.9
  4357.3  344.98  4421.3  342.44  4598.9  337.57  4784.5  335.81  4869.3  335.76
  4891.7  335.24  4905.1  336.14  4976.5  335.47  4990.9  334.44  4996.7  332.78
  5002.7  332.78  5003.9  332.02  5007.4  332.02    5011  335.35  5057.4  335.84
  5072.1  334.91  5082.3  335.38  5102.7  335.16  5123.1  336.56  5143.4  336.15
    5166  336.77  5194.4  335.78  5217.8  337.67  5306.4  340.11  5347.2   343.1
#Mann= 4 ,-1 , 0
  4186.9     .15       0  4282.8     .11       0  4976.5     .06       0
    5011     .11       0
Bank Sta=4976.5,5011
XS Rating Curve= 0 ,0
Exp/Cntr=0.3,0.1

Type RM Length L Ch R = 1 ,352000  ,663,663,663
BEGIN DESCRIPTION:
LAKE CREEK 682.0
END DESCRIPTION:
XS GIS Cut Line= 3
      3692217.86      10218311.1      3692004.04     10217806.86
      3691517.86     10217461.08
#Sta/Elev= 30
  4452.3   345.5  4484.9  345.35  4528.4  343.48  4572.5  342.45  4578.7  342.24
  4702.2  338.61  4725.3  338.64  4743.5  337.68  4886.8  335.94  4908.5  335.23
  4919.4   333.9  4928.9     332  4932.9     332  4949.2  334.13  4984.4334.2771
    4995  332.47    5000  332.24  5016.2  332.87 5022.35333.8882  5030.9  333.58
  5037.1  334.59  5123.2  333.67  5173.6   334.7  5216.2  333.88  5345.7  335.95
  5375.3  335.81    5438  336.99  5452.7  337.88  5517.9  339.43  5596.6  342.18
#Mann= 5 ,-1 , 0
  4452.3     .17       0  4572.5     .15       0  4578.7     .11       0
  4984.4     .06       0 5022.35     .11       0
Bank Sta=4984.4,5022.35
XS Rating Curve= 0 ,0
Exp/Cntr=0.3,0.1

Type RM Length L Ch R = 1 ,351337  ,276,276,276
BEGIN DESCRIPTION:
LAKE CREEK 681.0
END DESCRIPTION:
XS GIS Cut Line= 3
      3692717.83     10218261.04       3692073.8     10217331.13
      3691605.69      10217195.9
#Sta/Elev= 30
    3869  347.09  3998.7  343.82  4027.1  341.92  4076.4  340.98  4085.2  339.53
  4163.9  337.58  4250.4  336.68  4314.9  335.02  4329.8   336.6  4392.6  339.21
    4452  340.09  4601.4  334.08    4673  332.59  4723.7  333.04  4753.4  331.72
  4795.3  332.65  4947.3  331.67  4975.9  332.51  5000.2  330.24  5020.2  332.77
    5048   330.9  5057.2  328.32  5079.2   330.9  5087.4  332.59  5172.9  333.38
  5382.5  338.29  5410.9   339.6  5422.7  341.79  5449.7   339.3  5487.4  340.75
#Mann= 5 ,-1 , 0
    3869     .17       0  4163.9     .15       0  4250.4     .11       0
    5048     .06       0  5079.2     .11       0
Bank Sta=5048,5079.2
XS Rating Curve= 0 ,0
Exp/Cntr=0.3,0.1

Type RM Length L Ch R = 1 ,351061  ,784,784,784
BEGIN DESCRIPTION:
LAKE CREEK 680.0
END DESCRIPTION:
XS GIS Cut Line= 3
      3692797.74     10218075.89      3692250.88     10217143.63
      3691995.98     10216675.44
#Sta/Elev= 30
  3882.9   341.5  4039.2  336.69  4213.8  333.71  4266.7  333.82  4288.2  334.59
  4303.8  334.13  4331.1  335.21  4340.6  334.71  4426.9  335.55  4528.5  334.34
  4682.9  330.91    4763  331.65  4880.2  330.68  4982.1  331.62  5003.9  330.19
  5020.1  331.66  5047.6  330.84  5079.9  331.81  5091.9  330.81  5105.7  329.01
  5109.2  329.01  5114.6  330.66    5380  333.51  5423.7  334.54  5433.5  334.18
  5439.9  332.82    5456  331.29  5467.6  331.97  5477.9  334.74  5496.8  345.05
#Mann= 3 , 0 , 0
  3882.9     .11       0  5091.9     .06       0  5114.6     .11       0
Bank Sta=5091.9,5114.6
XS Rating Curve= 0 ,0
Exp/Cntr=0.3,0.1

Type RM Length L Ch R = 1 ,350277  ,468,468,468
BEGIN DESCRIPTION:
LAKE CREEK 679.0
END DESCRIPTION:
XS GIS Cut Line= 3
      3692867.85     10218111.03      3692834.21     10217174.88
      3692282.78     10216436.16
#Sta/Elev= 30
  4064.5  342.97  4254.6  338.18  4314.6  337.47    4486   332.3  4684.9  330.77
  4724.9  329.08    4825  328.33    4875  328.86    4925  328.24    4975  329.07
  4993.3  326.21  4996.8  326.21  5000.7  328.05  5016.3   328.5  5037.1  329.06
  5230.6  328.21  5251.8  328.96    5452  329.68  5587.5  328.91  5737.6  330.85
  5829.6  333.56  5837.6  333.41  5852.2  329.86  5858.5  329.92  5866.8  330.12
  5873.1  331.27  5887.7  336.05  5908.5  344.91  5916.9  346.55  5923.1  345.78
#Mann= 3 , 0 , 0
  4064.5     .11       0    4975     .06       0  5016.3     .11       0
Bank Sta=4975,5016.3
XS Rating Curve= 0 ,0
Exp/Cntr=0.3,0.1

Type RM Length L Ch R = 1 ,349809  ,309,309,309
BEGIN DESCRIPTION:
LAKE CREEK 678.0
END DESCRIPTION:
XS GIS Cut Line= 3
      3693094.63     10217919.66      3693235.26     10217060.29
      3693500.87     10215966.58
#Sta/Elev= 30
  4135.8  335.38    4256  332.97    4337  330.38  4478.9  328.62  4539.7  328.24
  4556.6  328.85  4671.4  328.95  4691.7  327.39  4722.1  327.82  4772.7  326.46
    4793  327.36  4863.4  328.14  4904.5  326.88  4924.7  328.12  4985.5  328.02
  4991.2  325.34  4993.1  323.85  4999.3  323.85  5003.7  325.68  5008.8  325.68
  5016.1     328  5273.4  329.04  5304.2  329.33  5324.8   330.3  5386.5  329.62
    5438  330.66  5468.9   330.2    5672  331.54  5849.6  334.17  6132.1  337.26
#Mann= 3 , 0 , 0
  4135.8     .11       0  4985.5     .06       0  5016.1     .11       0
Bank Sta=4985.5,5016.1
XS Rating Curve= 0 ,0
Exp/Cntr=0.3,0.1

Type RM Length L Ch R = 1 ,349500  ,500,500,500
BEGIN DESCRIPTION:
LAKE CREEK 677.0
END DESCRIPTION:
XS GIS Cut Line= 3
      3693271.71     10217956.13      3693501.34     10217178.32
      3693766.19     10216014.79
#Sta/Elev= 30
    4189  335.47  4229.6  334.91  4262.9  332.63  4268.1  334.03  4350.7   331.5
    4368  331.39  4373.2  332.07  4583.4  327.91  4616.7  326.24  4746.9  326.19
  4764.6  322.43  4778.2  322.96  4793.6  326.24  4809.5  326.98  4840.7  327.44
  4865.4  326.51  4898.7  327.44    4945  326.48  4976.3  326.85    5000  325.28
  5004.6  323.43  5017.7  326.85  5052.7  327.67  5192.1  326.25  5364.3  327.52
  5735.6  332.22  5848.4   332.2  5906.4  334.02  6166.3  337.18  6193.3  338.28
#Mann= 3 , 0 , 0
    4189     .11       0  4976.3     .06       0  5017.7     .11       0
Bank Sta=4976.3,5017.7
XS Rating Curve= 0 ,0
Exp/Cntr=0.3,0.1

Type RM Length L Ch R = 1 ,349000  ,500,500,500
BEGIN DESCRIPTION:
LAKE CREEK 676.0
END DESCRIPTION:
XS GIS Cut Line= 3
      3693969.63     10218117.62      3693919.67     10217333.61
      3693922.75     10216155.01
#Sta/Elev= 30
  4214.4  334.79  4331.2   332.4  4391.3   329.8  4794.9  325.74  4802.1  325.23
    4819  320.61  4825.3  320.61  4842.2  324.75  4862.3  325.93  4882.3  325.31
  4892.3  325.87  4902.3  324.91  4922.4  325.65  4962.5  324.55  4982.5  325.04
  4992.5  324.08  4998.8  322.11  5003.8  322.11  5022.5  325.82  5212.5  324.48
  5452.5     326  5662.5  328.55  5862.5  332.52  5902.5  332.36  5912.5  333.76
  5942.5     333  5982.5  333.73  6022.5  333.35  6072.5  335.51  6178.6     337
#Mann= 3 , 0 , 0
  4214.4     .11       0  4982.5     .06       0  5022.5     .11       0
Bank Sta=4982.5,5022.5
XS Rating Curve= 0 ,0
Exp/Cntr=0.3,0.1

Type RM Length L Ch R = 1 ,348500  ,614,614,614
BEGIN DESCRIPTION:
LAKE CREEK 675.0
END DESCRIPTION:
XS GIS Cut Line= 3
      3694017.84      10218111.1      3694263.49     10217172.31
      3694467.86     10216311.02
#Sta/Elev= 30
  4029.6   334.8  4143.3  331.14    4522  325.33  4608.5  325.28  4649.8  324.37
  4711.9  325.01  4815.2  323.94  4875.5  324.66  4921.1  323.82  4961.5  324.72
  4980.6  324.12  4990.9  323.09  4996.5  321.04  5003.5  321.04  5011.5  324.28
  5032.1  325.01  5062.9  323.95  5081.1  324.06  5086.2  325.03  5128.5  323.58
  5134.9  324.24  5196.5  323.92  5247.9  325.24  5339.5  325.94  5371.3  326.72
  5386.9  327.79  5434.2  328.71  5560.9  330.15  5771.9  334.35  5885.2  335.77
#Mann= 3 , 0 , 0
  4029.6     .11       0  4980.6     .06       0  5011.5     .11       0
Bank Sta=4980.6,5011.5
XS Rating Curve= 0 ,0
Exp/Cntr=0.3,0.1

Type RM Length L Ch R = 1 ,347886  ,386,386,386
BEGIN DESCRIPTION:
LAKE CREEK 674.0
END DESCRIPTION:
XS GIS Cut Line= 3
      3694500.88     10218117.55      3694537.34     10217643.63
      3694517.85     10216511.12
#Sta/Elev= 30
  4484.8   331.9    4742  326.64  4774.2  326.83  4842.3  324.98  4899.6  324.89
  4942.6  323.43  4982.7  323.27  4992.7  322.33  4999.2  318.74  5006.2  318.74
  5012.7  322.39  5022.7  323.15  5062.7  323.51  5092.7  322.95  5102.7  323.48
  5152.7  323.28  5162.7  322.42  5232.7  323.54  5242.7  322.98  5272.7  323.52
  5292.7  322.95  5412.7   323.8  5452.8  322.74  5482.8  319.88  5512.8  323.08
  5532.8  323.66  5602.8  323.62  5902.8  327.86  5982.8  330.33  6092.8  332.63
#Mann= 3 , 0 , 0
  4484.8     .11       0  4992.7     .06       0  5012.7     .11       0
Bank Sta=4992.7,5012.7
XS Rating Curve= 0 ,0
Exp/Cntr=0.3,0.1

Type RM Length L Ch R = 1 ,347500  ,500,500,500
BEGIN DESCRIPTION:
LAKE CREEK 673.0
END DESCRIPTION:
XS GIS Cut Line= 3
      3694767.85     10218161.05      3694855.35     10217497.09
      3694767.85     10216511.06
#Sta/Elev= 30
  4330.3   331.9  4572.4  328.51  4693.4  324.96  4743.8   324.1  4834.6  323.16
  4864.9  323.63  4935.5  321.93  4965.7  322.65  4980.9  321.98  4985.9  320.99
  4991.9  317.36  4999.1  317.36  5016.1  322.63  5106.4  322.31  5206.8  323.11
  5258.3     321  5297.2  323.74  5317.3  323.57  5337.3  320.08  5347.4  322.38
  5357.4  323.18  5377.5  322.88  5387.5  322.13  5407.6  322.83  5417.7  322.36
  5447.8  323.12  5598.6  324.52  5799.1   329.4  5909.6  331.09  5989.9  333.44
#Mann= 3 , 0 , 0
  4330.3     .11       0  4980.9     .06       0  5016.1     .11       0
Bank Sta=4980.9,5016.1
XS Rating Curve= 0 ,0
Exp/Cntr=0.3,0.1

Type RM Length L Ch R = 1 ,347000  ,294,294,294
BEGIN DESCRIPTION:
LAKE CREEK 672.0
END DESCRIPTION:
XS GIS Cut Line= 3
      3695579.01     10218331.14      3695126.87     10217107.93
      3694828.99     10216497.76
#Sta/Elev= 30
  3695.9  333.17  3962.5  327.42  4133.1  325.04    4264  324.31  4282.3  323.44
  4638.1   322.6  4718.6  321.45  4730.1  320.11  4740.8  321.41  4749.1   321.5
  4794.1  320.27    4835  321.23  4920.9  320.71  4956.6  321.31  4975.3  318.92
  4981.7  319.15    4987  317.73    5000  317.99    5002  315.94  5009.3  315.94
  5028.1  321.75  5033.7  319.26  5050.7  322.33  5085.5  322.22    5130  323.25
  5185.7  323.03  5354.6  325.28  5602.4     331  5641.9  332.84    5679  332.81
#Mann= 3 , 0 , 0
  3695.9     .11       0  4956.6     .06       0  5028.1     .11       0
Bank Sta=4956.6,5028.1
XS Rating Curve= 0 ,0
Exp/Cntr=0.3,0.1

Type RM Length L Ch R = 1 ,346706  ,206,206,206
BEGIN DESCRIPTION:
Mapping XS 2f667da0
END DESCRIPTION:
XS GIS Cut Line= 2
      3695740.47     10218466.57      3695245.67     10216581.12
#Sta/Elev= 30
  3563.1  335.96  3641.2  333.57  3692.8  333.13  3785.4     330    3831  331.11
  3878.9  330.19  3906.5  328.65  4027.7  326.68  4062.9  325.12  4143.6  325.19
  4323.5  322.51  4830.1  321.32  4912.8  319.25  4943.8  320.03  4970.8  318.19
    4976  319.72  4985.2  318.21  4991.8  314.41  4999.2  314.41 5007.38319.1331
  5011.2   321.8  5016.4  320.92  5026.5  321.94  5181.6  322.16    5316  326.51
  5336.7  328.63  5369.4  328.02  5485.4  333.77  5502.1   336.2  5512.4  335.69
#Mann= 4 ,-1 , 0
  3563.1     .11       0  4970.8     .08       0    4976     .06       0
 5007.38     .11       0
Bank Sta=4976,5007.38
XS Rating Curve= 0 ,0
Exp/Cntr=0.3,0.1

Type RM Length L Ch R = 1 ,346500  ,450,450,450
BEGIN DESCRIPTION:
LAKE CREEK 671.0
END DESCRIPTION:
XS GIS Cut Line= 3
      3695927.96     10218450.92      3695567.88     10217096.57
      3695454.27     10216514.76
#Sta/Elev= 30
  3598.6  334.89  3981.3  324.83  4105.5  322.83  4188.2  323.87  4197.8  322.41
    4203  323.65  4208.9   322.3  4229.6  321.35  4554.1  320.57  4798.7  322.03
  4840.1     321  4891.9   321.7  4912.6  319.87  4940.1  320.68    4954  319.65
  4985.4  320.86  4995.1  318.26    5000  318.26  5001.9  314.41  5009.3  314.41
  5023.6  320.53  5075.9  321.44  5081.4  321.68  5158.4   322.1  5183.3  321.09
  5321.5   325.7  5441.1  331.46  5497.8  332.49  5549.4  336.44  5592.8  337.65
#Mann= 5 ,-1 , 0
  3598.6     .11       0  4985.4     .06       0  5023.6     .11       0
  5075.9     .15       0  5081.4     .11       0
Bank Sta=4985.4,5023.6
XS Rating Curve= 0 ,0
Exp/Cntr=0.3,0.1

Type RM Length L Ch R = 1 ,346050  ,550,550,550
BEGIN DESCRIPTION:
LAKE CREEK 670.0
END DESCRIPTION:
XS GIS Cut Line= 4
      3695959.21     10218247.78      3695797.76     10217398.84
      3695943.59     10217159.25      3696058.17     10216601.95
#Sta/Elev= 30
  3969.2  328.72  4007.4  328.19  4047.3   323.6  4059.7  323.89    4088  327.64
  4118.5  324.36    4261  322.24  4320.7   322.8  4325.8  321.38  4393.4  320.35
  4627.5  320.11  4701.4  321.41  4739.5  320.11  4780.2  321.26  4842.8  320.02
  4977.4  320.18  5002.6  316.66  5010.1  316.66  5020.1  319.71  5029.7  320.58
  5072.5   320.5  5152.8  319.73    5164  318.43  5173.2  319.69  5244.7  319.79
  5285.5  321.75  5336.6  322.32    5551  328.74  5581.6  330.51  5682.8   331.8
#Mann= 5 ,-1 , 0
  3969.2     .11       0  4842.8     .15       0  4977.4     .09       0
  5029.7     .15       0  5072.5     .11       0
Bank Sta=4977.4,5029.7
XS Rating Curve= 0 ,0
Exp/Cntr=0.3,0.1

Type RM Length L Ch R = 1 ,345500  ,500,500,500
BEGIN DESCRIPTION:
LAKE CREEK 669.0
END DESCRIPTION:
XS GIS Cut Line= 3
      3696105.04     10218206.17      3696193.25     10217598.03
      3696117.85     10216761.02
#Sta/Elev= 30
  4385.5  327.67    4438  325.34  4633.2  321.02  4718.8  320.28  4744.3   319.4
  4976.7  317.58  4986.8  313.55  4990.8   310.2  4998.3   310.2  5003.2  318.33
  5008.2   314.8    5017  318.93  5027.8  318.81  5077.3  318.34  5097.4  319.04
  5114.2   317.5  5119.2  317.97  5157.5  317.16  5197.8  318.38  5341.1  319.32
  5358.4  318.74  5428.7  319.34  5438.7  318.63  5539.1  319.07  5569.3  320.58
  5609.4  321.38  5619.5  320.87  5668.9  322.64    5760  324.38  5840.4  327.21
#Mann= 5 ,-1 , 0
  4385.5     .11       0  4976.7     .07       0  5003.2     .11       0
  5027.8     .15       0  5157.5     .11       0
Bank Sta=4976.7,5003.2
XS Rating Curve= 0 ,0
Exp/Cntr=0.3,0.1

Type RM Length L Ch R = 1 ,345000  ,454,454,454
BEGIN DESCRIPTION:
LAKE CREEK 668.0
END DESCRIPTION:
XS GIS Cut Line= 3
      3696589.42     10218101.99      3696628.63     10217611.86
      3696443.59     10216518.61
#Sta/Elev= 30
  4508.3  325.58  4639.6  324.38    4760   319.6  4850.3  317.34  4976.2   317.6
  4980.7  317.73 4985.66316.6447  4990.8  315.52  4994.1   312.2  5010.9  312.84
 5022.35316.4339  5030.4  318.52  5035.4  317.59  5041.4   318.2  5095.8  317.72
  5123.9  313.66  5142.8  314.14  5151.2   316.1  5173.2   317.8  5203.6  317.12
  5355.8  317.85  5507.9  317.37  5538.3  319.12  5558.6  318.31  5781.7   320.4
  5815.4  321.76  5862.9  321.82  5875.8  323.09  5903.5   322.1  6108.8  327.36
#Mann= 5 ,-1 , 0
  4508.3     .11       0  4976.2     .15       0 4985.66     .09       0
 5022.35     .15       0  5123.9     .11       0
Bank Sta=4985.66,5022.35
XS Rating Curve= 0 ,0
Exp/Cntr=0.3,0.1

Type RM Length L Ch R = 1 ,344546  ,320,320,320
BEGIN DESCRIPTION:
LAKE CREEK 667.0
END DESCRIPTION:
XS GIS Cut Line= 3
      3696865.46     10218070.75      3696964.42     10217523.84
      3696657.14     10216518.65
#Sta/Elev= 30
  4436.5  323.41  4629.3  320.89    4741  317.56  4868.7  316.78  4893.5  316.71
  4913.8   317.3  4923.1  318.31  4964.6  317.62  4974.8  316.59  4981.7     314
  4986.8  314.63  4991.2  312.18  5001.8  311.15  5009.4  311.15  5016.1  314.05
  5026.6  316.53  5037.1  316.97  5047.5  314.02  5057.9  312.38  5068.9   314.9
  5078.8  316.23  5102.6  316.32  5110.2  317.08  5233.8  315.75  5648.2  317.92
  5882.9  321.52  5958.9  324.76  5986.5   323.2    5999  324.05  6043.4  324.71
#Mann= 5 ,-1 , 0
  4436.5     .11       0  4868.7     .15       0  4974.8     .09       0
  5026.6     .15       0  5068.9     .11       0
Bank Sta=4974.8,5026.6
XS Rating Curve= 0 ,0
Exp/Cntr=0.3,0.1

Type RM Length L Ch R = 1 ,344226  ,638,638,638
BEGIN DESCRIPTION:
Mapping XS 234237df
END DESCRIPTION:
XS GIS Cut Line= 3
      3696448.77     10218648.87      3697224.84     10217742.59
      3696829.06      10216445.9
#Sta/Elev= 30
  3718.9  335.31  3730.5  332.79    3759  331.23  3929.1  328.09  4412.1  323.67
  4510.9  320.89    4759  317.51  4851.2  317.58  4915.5     319  4924.1  317.58
  4997.3  316.22  5003.9  312.55  5011.5  312.55  5017.3  316.08  5022.5  317.09
  5045.1  316.85    5181  316.12  5295.5  316.32  5333.5  315.87  5342.3  314.29
  5352.8  314.09  5373.7  315.62  5457.3   316.8  5535.6  315.22  5561.9  316.39
  5568.4  315.45  5718.7  315.99  5983.1  320.66  6199.7  322.86  6267.8  324.63
#Mann= 5 ,-1 , 0
  3718.9     .11       0  4997.3     .06       0  5017.3     .11       0
  5045.1     .15       0    5181     .11       0
Bank Sta=4997.3,5017.3
XS Rating Curve= 0 ,0
Exp/Cntr=0.3,0.1

Type RM Length L Ch R = 1 ,343588  ,636,636,636
BEGIN DESCRIPTION:
Mapping XS 59c53da6
END DESCRIPTION:
XS GIS Cut Line= 4
      3696511.32      10218773.8      3697401.92     10217664.46
      3697308.17     10216893.63       3696896.7     10216440.49
#Sta/Elev= 30
  3084.1  332.48  3203.9  328.72  3410.3  325.36  3680.7  324.58    3916  320.86
  3922.4  319.63  3965.6  318.81    3980  321.01  3994.4  319.64  4064.8   318.2
  4256.8  317.09  4343.2  318.37  4424.2  316.99  4530.3  315.77  4626.2  316.28
  4973.5  315.87  4992.3  313.19  4992.9  308.14  4993.4  307.64  5001.2  307.64
  5003.7  311.75  5013.8  315.57    5074  314.99  5084.3  312.46  5108.5  313.64
  5165.8  315.36  5185.1  317.07    5349  315.35  5603.8  317.59  5895.3  324.02
#Mann= 6 ,-1 , 0
  3084.1     .11       0  4424.2     .17       0  4626.2     .15       0
  4973.5     .09       0  5013.8     .15       0  5108.5     .11       0
Bank Sta=4973.5,5013.8
XS Rating Curve= 0 ,0
Exp/Cntr=0.3,0.1
