HEC-RAS study LAKE CREEK.prj: LAKE CREEK Base Level Engineering

--- LAKE CREEK.g01 (geometry) --- (continued)

Type RM Length L Ch R = 1 ,342952  ,477,477,477
BEGIN DESCRIPTION:
Mapping XS 6c86430d
END DESCRIPTION:
XS GIS Cut Line= 4
      3696506.07     10218904.06      3697579.01     10217648.84
       3697636.3     10217091.54      3697042.68     10216372.95
#Sta/Elev= 30
  3105.2  333.42  3271.6   328.3  3519.7  324.09    3804  324.33  3902.8   321.8
  3924.8  322.96  3945.6  321.12  4009.3   319.9  4194.9  318.65  4295.3  317.48
  4498.9  316.33  4572.6   317.2  4661.1  315.44  4864.8   315.5  4890.7   314.4
  4985.1  312.66  4990.1  311.56  4991.6  308.53  5025.7  312.63  5055.8  314.83
  5100.2  315.06  5136.3  316.29  5334.5  315.09  5415.5  315.53  5479.6  314.15
    5693   314.7  5997.8   317.8  6232.3  323.28  6246.6   325.1  6248.8  327.78
#Mann= 11 ,-1 , 0
  3105.2     .11       0  4194.9     .17       0  4295.3     .11       0
  4572.6     .17       0  4661.1     .11       0  4890.7     .15       0
  4985.1     .09       0  5025.7     .15       0  5100.2     .11       0
  5334.5     .15       0  5479.6     .11       0
Bank Sta=4985.1,5025.7
XS Rating Curve= 0 ,0
Exp/Cntr=0.3,0.1

Type RM Length L Ch R = 1 ,342475  ,475,475,475
BEGIN DESCRIPTION:
LAKE CREEK 663.0
END DESCRIPTION:
XS GIS Cut Line= 3
      3699372.25     10219422.73      3698115.46     10217523.84
      3697067.85     10216311.07
#Sta/Elev= 30
       0  326.61   493.9   324.1     545  321.98  1179.9  318.68  1297.1  316.22
    1405  317.17  1598.1  315.71  2061.5  314.09  2148.5  313.93  2175.8  315.38
  2256.5  314.16  2412.6  314.88  2511.3     316  2554.1  315.06  2560.7   313.7
  2574.9   305.8  2582.6  306.61  2603.5  313.95  2611.1  314.85    2632  316.81
  2638.6  315.57  2674.7  315.78  2730.7  313.47    3029  315.19  3049.9  314.57
  3064.2  310.98  3071.8  311.04  3100.1   314.5  3454.6  315.97  3879.7  324.84
#Mann= 8 ,-1 , 0
       0     .11       0  1598.1     .15       0  2061.5     .11       0
  2175.8     .15       0  2412.6     .11       0  2560.7     .09       0
  2611.1     .15       0  2730.7     .11       0
Bank Sta=2560.7,2611.1
XS Rating Curve= 0 ,0
Exp/Cntr=0.3,0.1

Type RM Length L Ch R = 1 ,342000  ,495,495,495
BEGIN DESCRIPTION:
LAKE CREEK 662.0
END DESCRIPTION:
XS GIS Cut Line= 3
      3699037.36     10218846.78      3698062.84     10217031.75
      3697067.86     10216011.08
#Sta/Elev= 30
  2939.9   321.6    3558  319.03  3607.6  317.08    4193  315.72  4331.1  314.74
  4384.6  312.53  4603.8   314.5  4767.8  312.53    4861  313.72  4937.5   314.4
  4959.4   312.6  4975.6  306.01  4981.3  308.96  4983.6  304.08  4995.2  304.08
  4997.5  306.65    5004  305.42  5011.1  308.36  5018.1  306.09  5025.3  310.44
  5032.3   307.6  5039.4  310.87  5046.4  306.65  5053.6  311.71  5060.5  310.96
  5067.7  313.61  5187.6  312.75    5301  315.28  5725.4  315.18  6425.4  331.79
#Mann= 5 ,-1 , 0
  2939.9     .11       0    4861     .15       0  4959.4     .09       0
  5067.7     .15       0  5187.6     .11       0
Bank Sta=4959.4,5067.7
XS Rating Curve= 0 ,0
Exp/Cntr=0.3,0.1

Type RM Length L Ch R = 1 ,341505  ,505,505,505
BEGIN DESCRIPTION:
LAKE CREEK 661.0
END DESCRIPTION:
XS GIS Cut Line= 3
      3699042.56     10218805.11      3698454.01     10217044.67
      3697328.98     10216180.07
#Sta/Elev= 30
  3064.1  321.39  3505.3  319.22  3901.3  319.48  4421.3  315.68  4547.6  316.83
  4555.1  315.26    4574  314.58  4637.1  315.64  4700.3  313.26  4737.2  313.75
  4763.5  311.07  4776.5  313.01  4789.8  313.02  4839.8  313.82  4863.5  312.07
  4969.7  313.41  4984.2   309.8    4993  304.32  5004.6  304.32  5019.6  313.34
  5169.1  314.06  5218.9  310.74  5297.8  314.05    5350  313.87  5533.5  313.06
  5569.7  314.54  5625.9  313.19  5760.9  315.52  5818.9  314.16  6339.2  324.22
#Mann= 5 ,-1 , 0
  3064.1     .11       0  4789.8     .15       0  4969.7     .09       0
  5019.6     .15       0    5350     .11       0
Bank Sta=4969.7,5019.6
XS Rating Curve= 0 ,0
Exp/Cntr=0.3,0.1

Type RM Length L Ch R = 1 ,341000  ,538,538,538
BEGIN DESCRIPTION:
LAKE CREEK 660.0
END DESCRIPTION:
XS GIS Cut Line= 3
      3699813.38     10217216.54      3698717.95     10216883.63
      3697402.35     10216206.35
#Sta/Elev= 30
  3855.1  326.78  3975.8   323.2    4031  323.49  4058.6  320.93  4238.7  316.76
  4892.2  312.23  4955.1  314.12  4979.2  312.51    4988  308.68  4991.5  303.67
  5003.3  303.67  5011.1  305.82  5022.6   313.2  5099.8  312.83  5127.6  308.43
  5135.1  310.96  5180.1  312.94    5255  311.89  5416.3  312.86  5432.4  312.19
  5438.8  309.75  5448.9  309.13  5471.1  311.89  5515.8  313.56  5686.2  313.59
  5742.8  311.13    5798  313.26  5825.8  312.24  6147.1  315.72  6479.7  323.26
#Mann= 5 ,-1 , 0
  3855.1     .11       0  4892.2     .15       0  4979.2     .09       0
  5022.6     .15       0  5515.8     .11       0
Bank Sta=4979.2,5022.6
XS Rating Curve= 0 ,0
Exp/Cntr=0.3,0.1

Type RM Length L Ch R = 1 ,340462  ,213,213,213
BEGIN DESCRIPTION:
LAKE CREEK 659.0
END DESCRIPTION:
XS GIS Cut Line= 3
      3699907.17     10216950.93      3698584.21     10216523.84
      3697464.39     10216154.03
#Sta/Elev= 30
  3605.3  326.62  3825.3  319.94  3930.3  318.71  3946.4  316.12  4015.7  314.63
  4413.7  311.51  4528.3  312.33  4565.6   310.5  4620.5  311.68  4960.5  312.94
  4981.2  309.31  4987.3  305.76  4995.5  304.82  4996.3  302.45  5008.1  302.45
  5012.7  312.92  5075.9  310.74  5202.3  312.35  5233.9  310.27    5278  312.87
  5349.7  312.46  5368.3     311  5373.5  308.39  5391.8  310.77  5412.9   308.2
  5431.8   311.4    5455  310.15  5468.8  312.87  5760.4  314.84  6174.8   323.3
#Mann= 5 ,-1 , 0
  3605.3     .11       0  4620.5     .15       0  4960.5     .09       0
  5012.7     .15       0    5278     .11       0
Bank Sta=4960.5,5012.7
XS Rating Curve= 0 ,0
Exp/Cntr=0.3,0.1

Type RM Length L Ch R = 1 ,340249  ,866,866,866
BEGIN DESCRIPTION:
Mapping XS c6464f07
END DESCRIPTION:
XS GIS Cut Line= 4
      3699886.28     10216877.99      3698599.84     10216362.38
      3698422.76     10216456.13      3697491.67     10216071.21
#Sta/Elev= 30
  3741.4  325.62  3912.7  319.54  4014.9  318.68  4122.5  313.68  4636.7  311.68
  4690.2  310.05  4720.1  312.28  4967.9  312.74  4978.1  308.64  4983.5  302.16
  4995.3  302.16  5007.7  308.56  5021.7  311.82  5163.5  313.06  5239.6  309.64
  5299.3  312.26  5410.3  310.54  5442.7  312.05    5482  311.77  5511.3   307.9
  5527.8  307.86  5535.2  311.21  5549.4  312.32  5588.4  309.83  5617.8  312.53
  5711.7  312.23    5772  314.49  5825.3  313.34  5830.8  314.91  6335.2  323.91
#Mann= 5 ,-1 , 0
  3741.4     .11       0  4636.7     .15       0  4967.9     .09       0
  5021.7     .15       0  5442.7     .11       0
Bank Sta=4967.9,5021.7
XS Rating Curve= 0 ,0
Exp/Cntr=0.3,0.1

Type RM Length L Ch R = 1 ,339383  ,275,275,275
BEGIN DESCRIPTION:
LAKE CREEK 657.0
END DESCRIPTION:
XS GIS Cut Line= 3
      3699933.21     10216794.69      3698454.01     10216075.92
      3697351.34      10215571.4
#Sta/Elev= 30
  3359.4  326.07  3380.6  323.84  3397.6  324.78  3476.5  320.93    3702   317.6
  3814.7  312.75  4045.9  311.64  4113.6  313.06  4130.6  311.61  4235.6   311.4
  4246.1  311.26  4310.4  312.92    4341  311.83    4744  313.21  4959.3   310.4
  4981.9   305.4  4982.2  300.44  4982.7  299.94  4998.9  300.58  5003.8  304.73
  5021.8  307.28  5027.5  310.07    5033  311.59    5079  310.47  5115.1  312.32
  5235.7  311.82  5307.5  312.76  5406.7  312.56  5630.3  316.08  6216.6  332.85
#Mann= 9 ,-1 , 0
  3359.4     .11       0  4235.6     .15       0  4246.1     .11       0
    4341     .15       0  4959.3     .09       0  5027.5     .15       0
  5115.1     .11       0  5235.7     .15       0  5307.5     .11       0
Bank Sta=4959.3,5027.5
XS Rating Curve= 0 ,0
Exp/Cntr=0.3,0.1

Type RM Length L Ch R = 1 ,339108  ,689,689,689
BEGIN DESCRIPTION:
LAKE CREEK 656.0
END DESCRIPTION:
XS GIS Cut Line= 3
      3700302.94     10216659.24      3698313.38     10215763.42
      3697361.54     10215362.92
#Sta/Elev= 30
  3051.4  330.54    3355  325.79  3682.1  315.15  3914.7  311.44  4126.4  310.85
  4307.4  310.63  4388.3  310.63  4626.6   311.1  4650.1  311.14  4844.6  310.44
  4877.5  308.67  4930.7  311.61  4959.3  310.63  4965.2  306.87  4982.5  305.96
    4988  302.74  4998.1  301.96  4999.7  300.31  5011.5  300.31  5034.3  311.26
  5271.9  309.62  5462.1  312.54    5608  316.64  5637.2  316.12  5843.4  323.44
  5896.3  327.99    5920  325.66  5949.2  325.63  6020.4  329.76    6266  336.63
#Mann= 9 ,-1 , 0
  3051.4     .11       0  4126.4     .15       0  4307.4     .11       0
  4388.3     .15       0  4626.6     .11       0  4650.1     .15       0
  4959.3     .09       0  5034.3     .15       0  5462.1     .11       0
Bank Sta=4959.3,5034.3
XS Rating Curve= 0 ,0
Exp/Cntr=0.3,0.1

Type RM Length L Ch R = 1 ,338419  ,491,491,491
BEGIN DESCRIPTION:
LAKE CREEK 655.0
END DESCRIPTION:
XS GIS Cut Line= 3
      3700276.92     10216549.88      3698740.46     10215346.75
      3697912.96     10214946.01
#Sta/Elev= 30
  3081.1  328.21    3358  324.83  3571.4  318.76  3600.3  319.38  3621.1  317.87
  3993.4  310.72  4105.7  308.75  4176.3  310.89  4240.5  308.52  4261.3  310.11
  4447.5  309.09  4532.5  310.86  4731.4  308.96  4867.9   309.8  4932.1  308.06
  4967.4  309.54  4973.8  305.08  4981.9  306.56  4988.2  300.59  4996.8  299.78
  5008.6  299.78  5010.5  302.08  5017.1  301.69  5023.5   309.7  5046.6  311.56
  5099.8  312.43  5222.8  312.15  5336.7  311.67  5579.6  314.17    5952  323.25
#Mann= 5 ,-1 , 0
  3081.1     .11       0  3993.4     .15       0  4967.4     .09       0
  5023.5     .15       0  5222.8     .11       0
Bank Sta=4967.4,5023.5
XS Rating Curve= 0 ,0
Exp/Cntr=0.3,0.1

Type RM Length L Ch R = 1 ,337928  ,328,328,328
BEGIN DESCRIPTION:
LAKE CREEK 654.0
END DESCRIPTION:
XS GIS Cut Line= 3
      3700193.62     10216383.24      3699089.42     10215075.92
      3698157.09     10214353.02
#Sta/Elev= 30
  3288.5  325.46  3783.9  318.93  4053.1   310.1    4195   308.9  4393.7  309.59
  4457.4  307.45  4479.5  309.11  4500.3  307.74  4640.3  308.97  4724.3  309.84
  4869.5  310.02  4904.7  307.26  4933.3  309.73  4954.1  309.05  4976.1  307.06
  4982.7  302.29  4984.5  299.05  4996.4  299.05  4996.9  299.55    4997  301.57
  4999.6  303.69  5003.9  303.69  5011.9  309.76  5140.5   307.6  5300.7  309.29
  5381.3  309.06  5567.8  313.62  5604.2  312.58  5838.8  315.18  6179.5  317.29
#Mann= 9 ,-1 , 0
  3288.5     .11       0    4195     .15       0  4640.3     .11       0
  4724.3     .15       0  4954.1     .09       0  5011.9     .15       0
  5300.7     .11       0  5604.2     .15       0  5838.8     .11       0
Bank Sta=4954.1,5011.9
XS Rating Curve= 0 ,0
Exp/Cntr=0.3,0.1

Type RM Length L Ch R = 1 ,337600  ,591,591,591
BEGIN DESCRIPTION:
LAKE CREEK 653.0
END DESCRIPTION:
XS GIS Cut Line= 3
      3700467.88     10216661.11      3699318.59     10214857.17
      3698121.78     10214222.34
#Sta/Elev= 30
  2860.7  330.66  2925.9  330.65  2955.6  327.94  3004.6  328.63  3520.1  320.88
  3643.3  321.02    3984  311.67  4135.5  309.57    4287  309.36  4328.5   308.8
    4860  309.23  4888.3  306.67  4917.6  308.91  4969.2  309.46  4975.2  307.35
  4989.7  297.55  5001.6  297.55  5004.1  302.51  5011.8  309.14  5020.4  310.28
  5026.1  308.82  5312.6  308.01  5344.6  307.72  5441.9  310.57  5470.9  309.64
  5553.2  311.45  5751.1  311.92  5789.4  313.64  5987.3   313.5  6354.4  318.99
#Mann= 6 ,-1 , 0
  2860.7     .11       0    4287     .17       0  4328.5     .15       0
  4969.2     .09       0  5011.8     .15       0  5312.6     .11       0
Bank Sta=4969.2,5011.8
XS Rating Curve= 0 ,0
Exp/Cntr=0.3,0.1

Type RM Length L Ch R = 1 ,337009  ,604,604,604
BEGIN DESCRIPTION:
LAKE CREEK 652.0
END DESCRIPTION:
XS GIS Cut Line= 4
      3700422.73     10216377.97      3699557.67     10215039.25
       3699761.3     10214559.43      3698292.69     10213832.27
#Sta/Elev= 30
  2783.8  325.62  3407.6  316.77  3443.9  319.15  3449.8  317.13    3471  316.12
  3610.1  312.06  3800.4  310.75  4072.6  308.29  4127.2  309.51  4254.1  306.89
  4304.1  309.59  4420.6  309.74  4620.7  307.63  4679.9  304.77  4702.6  307.37
  4974.7  308.68  4991.6  306.38  4997.3  297.71  5009.2  297.71  5025.5  308.57
  5192.9  306.76    5291  308.65  5339.1  312.05    5356  311.86    5384   307.5
  5445.7  306.62  5473.7  308.68  5594.6  310.39  6303.5  312.09  6537.7  317.36
#Mann= 6 ,-1 , 0
  2783.8     .11       0  3800.4     .17       0  4127.2     .15       0
  4974.7     .09       0  5025.5     .15       0    5291     .11       0
Bank Sta=4974.7,5025.5
XS Rating Curve= 0 ,0
Exp/Cntr=0.3,0.1

Type RM Length L Ch R = 1 ,336405  ,405,405,405
BEGIN DESCRIPTION:
LAKE CREEK 651.0
END DESCRIPTION:
XS GIS Cut Line= 3
      3701375.05      10215155.8      3699977.44     10214235.64
      3698562.71      10213411.1
#Sta/Elev= 30
  3374.7  323.42  3844.2  314.32  3896.9     314  3923.9  319.49  3938.8  319.12
  3960.1  315.23  4074.7  313.77  4251.4  312.97  4535.7  308.92  4586.3  308.75
  4766.2  307.85  4776.2  308.01  4856.7  307.15  4920.9  306.81  4941.9  302.44
  4978.1  307.96  4987.2   304.1  4993.6  297.16  5005.7  297.16  5008.2  301.35
  5023.3  306.88  5333.5  307.63  5386.9  307.86  5417.9  311.31  5461.3  307.61
  5547.3  307.25  5578.8  311.78    5659  307.93    6205  309.73  6685.5  315.84
#Mann= 13 ,-1 , 0
  3374.7     .11       0  3844.2     .15       0  3938.8     .11       0
  4074.7     .17       0  4251.4     .11       0  4535.7     .15       0
  4586.3     .11       0  4766.2     .17       0  4776.2     .11       0
  4856.7     .15       0  4978.1     .09       0  5023.3     .15       0
  5333.5     .11       0
Bank Sta=4978.1,5023.3
XS Rating Curve= 0 ,0
Exp/Cntr=0.3,0.1

Type RM Length L Ch R = 1 ,336000  ,500,500,500
BEGIN DESCRIPTION:
LAKE CREEK 650.0
END DESCRIPTION:
XS GIS Cut Line= 3
      3701017.82     10214611.05      3700050.16     10213957.84
      3698067.83     10212561.06
#Sta/Elev= 30
  3832.5  318.39  4328.6  308.91  4648.8  307.76  4826.1  304.07  4877.1  307.68
    4970  307.44    4985  304.58  4992.3  297.07  5004.4  297.07    5006  301.82
  5020.8  307.74  5172.3  306.69  5199.4  303.59  5235.3   307.6  5528.8  307.81
  5726.7  308.36  5844.3  309.41  5850.8  309.26  6058.2  310.36  6284.5  309.04
  6305.4  312.48  6320.2  309.37  6456.9  313.99  6477.8  310.03  6519.7  313.25
  6570.2  310.65  6667.1   313.7  6871.5  315.23  7226.3  320.18    7425  323.23
#Mann= 12 ,-1 , 0
  3832.5     .11       0  4648.8     .15       0    4970     .09       0
  5020.8     .15       0  5528.8     .11       0  5726.7     .17       0
  5844.3     .11       0  5850.8     .17       0  6058.2     .15       0
  6667.1     .11       0  6871.5     .15       0  7226.3     .11       0
Bank Sta=4970,5020.8
XS Rating Curve= 0 ,0
Exp/Cntr=0.3,0.1

Type RM Length L Ch R = 1 ,335500  ,276,276,276
BEGIN DESCRIPTION:
LAKE CREEK 649.0
END DESCRIPTION:
XS GIS Cut Line= 3
      3701067.88      10214561.1      3700277.02     10213624.16
      3698717.88     10212661.09
#Sta/Elev= 30
  3773.9  318.64  4401.3  307.07  4526.3  307.05  4575.6  307.45  4589.8  303.65
  4628.4  307.26  4823.9   304.8  4959.1  307.26  4973.4  305.92  4988.2  295.32
  5000.3  295.32  5010.1   303.1    5016  302.53  5022.5  307.14    5126  306.65
  5168.5  303.86  5183.9  306.25  5220.6  307.09  5305.7  306.94  5363.6  304.25
  5415.6  306.81  5594.3  306.74  5634.4   307.6  5832.8  309.46  6010.3  308.39
  6272.8  310.28    6626  316.97  6641.4  317.47  6715.4  318.84  6832.6  320.09
#Mann= 12 ,-1 , 0
  3773.9     .11       0  4401.3     .17       0  4526.3     .11       0
  4628.4     .15       0  4959.1     .09       0  5022.5     .15       0
  5594.3     .17       0  5634.4     .15       0  5832.8     .17       0
    6626     .15       0  6641.4     .17       0  6715.4     .11       0
Bank Sta=4959.1,5022.5
XS Rating Curve= 0 ,0
Exp/Cntr=0.3,0.1

Type RM Length L Ch R = 1 ,335224  ,738,738,738
BEGIN DESCRIPTION:
LAKE CREEK 648.0
END DESCRIPTION:
XS GIS Cut Line= 3
      3701114.62     10214079.41      3700246.54     10213332.86
      3698767.84     10212661.07
#Sta/Elev= 30
  4045.6   314.6  4413.5  306.97  4743.9  305.88  4760.5   304.5    4801  306.33
  4956.8  306.24  4964.5  305.01  4971.1  300.77  4985.8  295.89    4998  295.89
  5006.2  302.09  5013.8  298.59  5020.4  305.04  5028.1   304.1  5034.7  306.78
  5176.3  306.51  5229.3  301.62    5266  305.72  5407.9  305.39  5430.7  303.11
  5476.5  306.17  5522.7  304.65  5540.3  306.46  5608.9  306.09  5715.4  306.94
  5947.6  308.55  6052.2  310.82  6340.1  310.77  6739.2  318.93  6814.7  319.86
#Mann= 10 ,-1 , 0
  4045.6     .11       0  4413.5     .17       0  4760.5     .15       0
  4956.8     .09       0  5034.7     .15       0  5407.9     .17       0
  5608.9     .15       0  5715.4     .11       0  5947.6     .17       0
  6739.2     .11       0
Bank Sta=4956.8,5034.7
XS Rating Curve= 0 ,0
Exp/Cntr=0.3,0.1

Type RM Length L Ch R = 1 ,334486  ,486,486,486
BEGIN DESCRIPTION:
LAKE CREEK 647.0
END DESCRIPTION:
XS GIS Cut Line= 3
      3701317.82     10214161.03      3700602.44     10213098.49
      3698667.83     10212561.06
#Sta/Elev= 30
  3848.4  317.16  4281.7   311.3  4416.7  307.14  4439.1  308.34  4468.8  314.36
  4503.6  310.68  4733.9  305.31  4855.5  303.02  4908.5   304.8  4929.5  302.55
  4950.5  304.86  4971.5  304.54  4980.4  303.33  4986.5  300.03    4987  295.05
  4987.5  294.55  4999.7  294.55  5016.4   304.1  5022.5  306.04  5043.5  306.85
  5109.4  305.25  5619.8  304.26    5782  304.79  5875.7  305.55  6086.1  306.61
  6187.5  308.25  6216.1   308.7  6489.9  311.75  6618.2   312.1  7137.2  319.76
#Mann= 13 ,-1 , 0
  3848.4     .11       0  4468.8     .17       0  4733.9     .11       0
  4855.5     .15       0  4971.5     .09       0  5016.4     .15       0
  5619.8     .17       0    5782     .11       0  5875.7     .15       0
  6086.1     .17       0  6187.5     .11       0  6216.1     .17       0
  6489.9     .11       0
Bank Sta=4971.5,5016.4
XS Rating Curve= 0 ,0
Exp/Cntr=0.3,0.1

Type RM Length L Ch R = 1 ,334000  ,500,500,500
BEGIN DESCRIPTION:
LAKE CREEK 646.0
END DESCRIPTION:
XS GIS Cut Line= 3
      3701366.34     10214009.98      3700907.77     10212931.31
       3699291.4     10212689.18
#Sta/Elev= 30
  3827.9  314.41  4274.5  309.58  4374.5  311.51  4474.5  308.55  4627.3  306.25
  4772.9  306.45  4838.2  303.76  4924.2   305.2  4961.8  304.47  4967.7  301.78
  4985.5  301.71  4991.3  294.17  5003.5  294.17  5020.1  304.07  5030.3  305.19
  5040.4  303.74  5070.7  305.37  5237.7  305.77  5313.4  303.98  5363.9  305.21
    5743  304.29  5893.8  304.62  5990.9  304.03  6047.2  305.83  6122.3  305.31
  6223.4   307.7  6336.5  307.39    6521   311.5  6565.9  311.19  6634.4  312.23
#Mann= 8 ,-1 , 0
  3827.9     .11       0  4772.9     .15       0  4961.8     .09       0
  5020.1     .15       0    5743     .17       0  5893.8     .15       0
  6336.5     .17       0  6565.9     .11       0
Bank Sta=4961.8,5020.1
XS Rating Curve= 0 ,0
Exp/Cntr=0.3,0.1

Type RM Length L Ch R = 1 ,333500  ,500,500,500
BEGIN DESCRIPTION:
LAKE CREEK 645.0
END DESCRIPTION:
XS GIS Cut Line= 4
      3701479.19     10214070.74      3701089.49     10212701.98
      3700769.11      10212681.3      3699178.81     10212655.78
#Sta/Elev= 30
  3255.8  315.32  3756.7  309.67  3936.4  310.64  4009.3  308.38  4253.6  307.42
  4399.2  304.27  4629.6  304.07  4713.9  303.92  4804.1  303.91    4891  306.21
  4981.2  304.09  4991.2  298.93  4991.5  294.49    4992  293.99  5004.2  293.99
  5031.3  304.63  5051.3  305.52  5131.3     303  5201.3  303.06  5231.3  301.22
  5271.3  303.27  5351.3  304.17  5552.4  302.43  5746.1  304.59  5991.4  304.93
  6061.4  307.15  6180.4  307.45  6333.9  310.67  6491.4  313.17  6590.5  312.67
#Mann= 10 ,-1 , 0
  3255.8     .11       0  4629.6     .15       0  4713.9     .11       0
  4804.1     .15       0  4981.2     .09       0  5031.3     .15       0
  5552.4     .17       0  5746.1     .15       0  6180.4     .17       0
  6333.9     .11       0
Bank Sta=4981.2,5031.3
XS Rating Curve= 0 ,0
Exp/Cntr=0.3,0.1

Type RM Length L Ch R = 1 ,333000  ,504,504,504
BEGIN DESCRIPTION:
LAKE CREEK 644.0
END DESCRIPTION:
XS GIS Cut Line= 3
      3702720.54      10212603.7      3700759.28      10212335.6
      3699204.83      10212603.7
#Sta/Elev= 30
  3020.5  324.37  3194.8  319.93  3386.6  310.83  3598.6  307.35  4029.5  306.79
  4133.4  306.44  4181.6  303.01  4234.1  304.67  4258.9  302.76  4338.2  305.67
  4981.3  303.79  4991.3  302.37  4996.5   296.1  5004.6   296.9  5004.9  293.96
  5005.4  293.46  5021.7  294.06    5042  303.97  5052.2  305.72  5163.8  303.83
  5194.3  299.36  5224.7  303.68  5671.2  302.15  5752.4  305.25  5924.9   304.6
  6087.2  307.67  6158.3  306.09  6399.3  310.89  6462.7  313.12  6577.4  312.31
#Mann= 7 ,-1 , 0
  3020.5     .11       0  4029.5     .15       0  4234.1     .11       0
  4338.2     .15       0  4981.3     .09       0    5042     .15       0
  6399.3     .11       0
Bank Sta=4981.3,5042
XS Rating Curve= 0 ,0
Exp/Cntr=0.3,0.1

Type RM Length L Ch R = 1 ,332496  ,822,822,822
BEGIN DESCRIPTION:
LAKE CREEK 643.0
END DESCRIPTION:
XS GIS Cut Line= 3
      3702677.08     10212542.93      3700958.35     10212013.42
      3699213.55     10212499.53
#Sta/Elev= 30
  3331.7  323.48  3498.3  315.53  3770.4  308.62  4695.9  303.83    4733  302.04
    4754  303.86  4973.7  304.69 4976.11303.1839  4982.1  299.44  4987.3  300.68
  4994.6  295.64  5005.1  293.87  5014.8  295.53  5019.8  292.41  5032.2  292.41
  5036.5   296.5  5052.7  303.49  5431.7  303.94  5516.3  300.95  5535.5  303.51
  5702.9  303.42  5722.4  301.59  5731.9  303.47  5763.9  300.87  5776.5  302.95
  5805.4  301.42  5889.4   304.1  6336.2  304.28  6591.2  309.56  6941.4  313.02
#Mann= 4 ,-1 , 0
  3331.7     .11       0  4695.9     .15       0 4976.11     .09       0
  5052.7     .15       0
Bank Sta=4976.11,5052.7
XS Rating Curve= 0 ,0
Exp/Cntr=0.3,0.1

Type RM Length L Ch R = 1 ,331674  ,674,674,674
BEGIN DESCRIPTION:
LAKE CREEK 642.0
END DESCRIPTION:
XS GIS Cut Line= 3
      3702763.92     10212568.99      3701071.19     10211509.95
      3699067.84     10212461.08
#Sta/Elev= 30
  2867.3  325.11    3400   309.5  4473.4  301.13  4502.3  299.39  4516.5  301.98
  4547.6  302.65  4610.1   303.8    4863  301.71  4966.7  303.04  4978.4  302.85
  4994.4  292.84  5006.8  292.84  5017.7  302.38  5033.8  302.47  5421.2  301.38
  5443.4  298.77    5543  303.45  5551.5  300.72    5557  301.86  5574.2  298.29
    5597  301.98  5619.7  302.75  5720.2  303.21  6084.4  305.77  6164.6  305.78
  6306.8  309.72  6420.1  308.99  6908.5   313.1    6971  315.32  7081.7  314.45
#Mann= 8 ,-1 , 0
  2867.3     .11       0  4473.4     .15       0  4547.6     .11       0
  4610.1     .15       0  4966.7     .09       0  5033.8     .15       0
  5720.2     .11       0  6084.4     .15       0
Bank Sta=4966.7,5033.8
XS Rating Curve= 0 ,0
Exp/Cntr=0.3,0.1

Type RM Length L Ch R = 1 ,331000  ,500,500,500
BEGIN DESCRIPTION:
LAKE CREEK 640.0
END DESCRIPTION:
XS GIS Cut Line= 3
      3702717.88     10212461.09      3700799.76     10211035.12
      3699817.82     10210611.06
#Sta/Elev= 30
  2609.9  322.82  2953.1  313.25  3188.8   311.8    3389  306.69  3645.6  305.64
  3689.4  304.16  4025.2  301.57  4181.7  302.74  4210.9  297.61  4231.7  301.48
  4267.2  302.58  4553.8  300.85  4753.2  301.05  4776.2   302.6  4832.1  301.37
  4968.1  301.89  4982.7  301.66  4989.9  299.53  4997.3  294.61  5006.6  293.13
  5019.3  293.13  5026.1  299.72  5073.1  301.74  5125.5   300.1    5149  301.99
  5426.5  301.79  5590.3   302.3  5612.1  303.74  5749.7  305.37  6069.6  312.86
#Mann= 6 ,-1 , 0
  2609.9     .11       0  4832.1     .15       0  4989.9     .09       0
  5026.1     .15       0  5426.5     .17       0  5749.7     .11       0
Bank Sta=4989.9,5026.1
XS Rating Curve= 0 ,0
Exp/Cntr=0.3,0.1

Type RM Length L Ch R = 1 ,330500  ,587,587,587
BEGIN DESCRIPTION:
LAKE CREEK 639.0
END DESCRIPTION:
XS GIS Cut Line= 3
      3702867.88      10212561.1       3700992.1     10210664.39
      3699967.86     10210411.07
#Sta/Elev= 30
  2332.4  328.36  2855.7  314.83  3364.8  306.05  3831.5  303.66  3937.6  301.47
  4258.7  301.07  4329.9  301.12  4361.9  298.05    4376   301.2  4708.4  299.14
  4804.5  301.09    4970  301.66  4984.8  291.66  4997.5  291.66    4998  292.16
  4998.3   295.7  5004.8  296.68  5014.7  302.08  5120.4  300.84  5138.3  298.05
  5148.6  298.38  5156.7  300.75  5161.8  298.96  5169.2  300.68  5198.1  301.05
  5239.5  298.63  5261.9  300.89  5345.6  300.89  5931.2   307.9  6055.1   308.9
#Mann= 8 ,-1 , 0
  2332.4     .11       0  4258.7     .15       0  4329.9     .11       0
  4804.5     .15       0    4970     .09       0  5014.7     .15       0
  5345.6     .17       0  5931.2     .11       0
Bank Sta=4970,5014.7
XS Rating Curve= 0 ,0
Exp/Cntr=0.3,0.1

Type RM Length L Ch R = 1 ,329913  ,437,437,437
BEGIN DESCRIPTION:
LAKE CREEK 638.0
END DESCRIPTION:
XS GIS Cut Line= 3
      3702659.76     10211909.28      3701418.42     10210338.07
      3700388.54     10209755.57
#Sta/Elev= 30
  3097.6  314.07  3183.8  310.78  3496.3  305.81  3901.9  303.62  4030.1  304.14
  4165.8  301.84  4286.6  301.68  4350.7  299.92  4553.7  299.95  4671.3  300.33
  4749.9  297.99  4892.3  298.92  4963.1   300.9  4977.5  299.87    4992  296.31
    5000  291.75  5012.7  291.75  5027.2  300.89  5215.5  301.11  5385.3  298.83
  5723.8  298.61  5870.3  299.91  5913.6  302.31    6029  303.72  6051.1  304.64
  6156.1  306.69  6169.1  307.92  6249.5  307.28  6258.6  308.45  6283.2  314.81
#Mann= 7 ,-1 , 0
  3097.6     .11       0  4553.7     .15       0  4977.5     .09       0
  5027.2     .15       0  5723.8     .11       0    6029     .15       0
  6051.1     .11       0
Bank Sta=4977.5,5027.2
XS Rating Curve= 0 ,0
Exp/Cntr=0.3,0.1

Type RM Length L Ch R = 1 ,329476  ,243,243,243
BEGIN DESCRIPTION:
LAKE CREEK 637.0
END DESCRIPTION:
XS GIS Cut Line= 3
      3702763.93     10210980.46      3701678.83     10210207.86
      3700448.68     10209666.62
#Sta/Elev= 30
  3890.8  307.72  4031.7  307.59  4395.1  302.13  4616.8  300.64  4818.9  298.93
  4855.8  299.85  4919.4  298.17  4934.2  299.32  4963.7   299.1  4978.5  296.02
  4984.5  290.67  4997.2  290.67  5020.3  299.51  5027.6  301.42  5055.9  299.65
  5121.1  300.89  5162.9  299.49  5171.5  300.58  5379.3  299.58    5426  300.56
  5501.5  299.32  5600.3  299.96  5861.7  298.22  6116.4  299.12  6283.7  302.11
  6305.5  303.75  6343.5  303.32  6502.2  308.08  6534.9  306.74  6566.8  314.25
#Mann= 8 ,-1 , 0
  3890.8     .15       0  4395.1     .11       0  4616.8     .15       0
  4963.7     .09       0  5020.3     .15       0  5861.7     .17       0
  6116.4     .15       0  6343.5     .11       0
Bank Sta=4963.7,5020.3
XS Rating Curve= 0 ,0
Exp/Cntr=0.3,0.1

Type RM Length L Ch R = 1 ,329233  ,733,733,733
BEGIN DESCRIPTION:
LAKE CREEK 636.0
END DESCRIPTION:
XS GIS Cut Line= 3
      3703319.41     10210641.88      3701774.32     10210068.97
      3700582.53     10209479.93
#Sta/Elev= 30
  3477.7  313.01  3727.3  307.48  4368.3   301.9  4377.4     302  4630.7  299.98
  4726.6  300.97  4743.5   299.7  4762.3  299.08  4787.3  294.54  4812.4  299.56
  4887.2  298.91  4983.2  300.65  4989.3   293.7  4998.2  291.48  5010.9  291.48
  5014.4  295.58  5019.7  296.59  5025.8  300.13  5247.5  299.23  5277.8  298.11
  5623.3  298.67  5746.7  297.16  6082.4  299.43  6150.6  299.91  6266.1  303.01
  6327.1  305.26  6359.8  306.74  6419.9  305.58  6435.2  307.71    6455  313.83
#Mann= 11 ,-1 , 0
  3477.7     .15       0  4368.3     .11       0  4377.4     .15       0
  4630.7     .17       0  4743.5     .15       0  4983.2     .09       0
  5025.8     .15       0  6082.4     .17       0  6266.1     .11       0
  6327.1     .17       0  6435.2     .11       0
Bank Sta=4983.2,5025.8
XS Rating Curve= 0 ,0
Exp/Cntr=0.3,0.1

Type RM Length L Ch R = 1 ,328500  ,500,500,500
BEGIN DESCRIPTION:
LAKE CREEK 635.0
END DESCRIPTION:
XS GIS Cut Line= 3
      3703640.64     10210546.41      3702121.14     10209594.02
      3701089.43     10208739.09
#Sta/Elev= 30
  3206.7  321.04  3409.6  316.58  3436.7  317.26  3453.9  315.77  3574.5  311.21
    3593  310.53  3771.4  305.62  4109.7  301.98  4272.2  298.35  4335.5  298.79
  4368.5  298.59  4545.2  298.38  4662.4  297.71  4735.4  299.09  4756.6  296.82
  4779.6  298.48  4975.8  298.43  4991.2  294.61  4997.1  291.56  5005.2  291.05
  5018.1  291.05  5025.9     299    5289  297.27  5565.1  298.35  5643.2  296.99
  5757.5  298.99  5835.4   297.6  6173.5  298.63  6303.5  302.37  6339.9  311.26
#Mann= 11 ,-1 , 0
  3206.7     .17       0  3453.9     .15       0  3574.5     .17       0
    3593     .15       0  4109.7     .17       0  4335.5     .15       0
  4368.5     .17       0  4545.2     .15       0  4975.8     .09       0
  5025.9     .15       0  6173.5     .11       0
Bank Sta=4975.8,5025.9
XS Rating Curve= 0 ,0
Exp/Cntr=0.3,0.1

Type RM Length L Ch R = 1 ,328000  ,406,406,406
BEGIN DESCRIPTION:
LAKE CREEK 634.0
END DESCRIPTION:
XS GIS Cut Line= 3
        3703632.     10209947.47      3702458.23     10209299.61
      3701343.05     10208395.86
#Sta/Elev= 30
  3659.3  318.15    3682  318.55  4116.3  303.04  4309.7  300.14  4653.8  296.65
  4794.7   297.9  4806.3  295.96  4941.4  299.24  4973.1298.0438  4977.6  297.48
    4985   291.3  4990.7  293.33  4999.8  290.01  5012.7  290.01  5013.4  291.75
  5020.6  294.82  5027.1  293.04    5035  296.34  5049.4  298.03  5226.9  297.88
  5283.7  295.88  5447.4  297.37  5773.6  297.25  5810.3  295.82  5831.1  297.61
  6136.5  295.15  6246.9  299.41  6369.9  304.33  6414.5  305.24  6435.4  308.52
#Mann= 6 ,-1 , 0
  3659.3     .17       0  4309.7     .15       0  4973.1     .09       0
  5049.4     .15       0  6246.9     .11       0  6369.9     .17       0
Bank Sta=4973.1,5049.4
XS Rating Curve= 0 ,0
Exp/Cntr=0.3,0.1

Type RM Length L Ch R = 1 ,327594  ,594,594,594
BEGIN DESCRIPTION:
LAKE CREEK 633.0
END DESCRIPTION:
XS GIS Cut Line= 3
      3703567.88     10209811.09      3702590.29      10208940.5
      3701617.85     10208161.07
#Sta/Elev= 30
  3708.6  316.03  3930.6  307.93    4148  301.48  4473.3  299.93  4498.2  298.28
  4572.8  296.21  4643.8  296.77  4664.7  293.47  4686.1  296.73  4764.2  298.28
  4848.7  296.81    4934  298.66 4974.35 297.273  4983.3   293.1  4983.9  288.89
  4984.4  288.39  4997.3  288.39  5011.7  297.21  5021.2  298.61  5238.8  297.44
  5261.2     296    5282  297.08  5310.8  295.59  5339.6  296.92  5509.3  295.43
  5808.6  297.01  6050.2  295.23  6064.6  293.81  6159.9  301.41  6263.9   307.5
#Mann= 7 ,-1 , 0
  3708.6     .17       0  3930.6     .15       0  4473.3     .17       0
  4498.2     .15       0 4974.35     .09       0  5011.7     .15       0
  6159.9     .11       0
Bank Sta=4974.35,5011.7
XS Rating Curve= 0 ,0
Exp/Cntr=0.3,0.1

Type RM Length L Ch R = 1 ,327000  ,500,500,500
BEGIN DESCRIPTION:
LAKE CREEK 632.0
END DESCRIPTION:
XS GIS Cut Line= 3
      3703517.88     10209311.09       3702558.2     10208495.86
      3701567.87     10207961.08
#Sta/Elev= 30
  3740.8  306.98  3946.8  300.54  4194.7  296.34  4457.5  296.82  4492.6   292.5
  4500.4  296.36  4528.1  295.27    4596  296.62  4909.2  296.86  4968.2  296.92
  4982.5  290.23  4989.1  291.13  4993.4  288.54  5011.8  289.51 5032.98296.8673
  5122.8  297.65    5276  295.03  5439.7  296.02  5543.5  293.93  5587.3  296.01
  5794.8  294.01    5818  296.13  5920.4   303.9  5986.1  307.13  6035.5     305
  6073.6  308.69  6080.1     307  6089.8  307.24  6111.7  314.01  6125.5  313.29
#Mann= 7 ,-1 , 0
  3740.8     .17       0  4194.7     .15       0    4596     .17       0
  4909.2     .15       0  4968.2     .09       0 5032.98     .15       0
    5818     .11       0
Bank Sta=4968.2,5032.98
XS Rating Curve= 0 ,0
Exp/Cntr=0.3,0.1

Type RM Length L Ch R = 1 ,326500  ,500,500,500
BEGIN DESCRIPTION:
LAKE CREEK 631.0
END DESCRIPTION:
XS GIS Cut Line= 3
      3703667.88      10209161.1      3702702.34     10208207.03
      3701867.88     10207211.11
#Sta/Elev= 30
  3642.6  309.76  3925.5  300.25  4134.8  296.58  4314.4  294.74  4413.4  296.77
  4448.7  293.31    4477  296.64  4715.2  294.92  4850.8  295.09  4986.2  296.17
  4993.2  289.05  5006.1  289.05  5014.5  293.84 5026.46 296.207  5341.1  294.94
  5398.3  292.21  5447.8  295.65  5490.5   293.8  5568.8   295.3  5632.5   293.6
  5850.7  296.65  5901.9  296.87  5997.6  301.19  6037.2   302.5  6051.5  305.43
  6064.5  303.67  6078.9  304.93  6144.5  310.53  6190.7  313.78  6299.3  322.62
#Mann= 11 ,-1 , 0
  3642.6     .17       0  4134.8     .15       0  4715.2     .17       0
  4850.8     .15       0  4986.2     .09       0 5026.46     .15       0
  5850.7     .11       0  5997.6     .17       0  6078.9     .11       0
  6144.5     .17       0  6190.7     .11       0
Bank Sta=4986.2,5026.46
XS Rating Curve= 0 ,0
Exp/Cntr=0.3,0.1

Type RM Length L Ch R = 1 ,326000  ,429,429,429
BEGIN DESCRIPTION:
LAKE CREEK 630.0
END DESCRIPTION:
XS GIS Cut Line= 3
      3703917.81     10208511.05      3703137.25     10208003.25
      3702117.84     10207161.06
#Sta/Elev= 30
  4068.8  309.01  4169.9  305.65  4227.2   306.7    4776  295.56  4891.9  293.59
  4978.9  295.95  4990.9  287.79  5003.9  287.79  5008.5  291.95    5015  289.65
  5022.8  294.99  5029.3  293.39  5037.2  296.19  5206.8  293.85  5321.2   295.2
  5356.3  293.09  5377.1  294.75  5519.1  294.73    5583  294.08  5611.6  291.85
  5619.5  293.33  5683.3  294.51  6037.6  293.56  6179.6  299.39  6222.6  303.71
  6244.5  301.56  6255.2  304.35    6280  303.95  6294.3  306.27  6322.3  306.62
#Mann= 5 ,-1 , 0
  4068.8     .17       0    4776     .15       0  4978.9     .09       0
  5037.2     .15       0  6255.2     .11       0
Bank Sta=4978.9,5037.2
XS Rating Curve= 0 ,0
Exp/Cntr=0.3,0.1

Type RM Length L Ch R = 1 ,325571  ,571,571,571
BEGIN DESCRIPTION:
LAKE CREEK 629.0
END DESCRIPTION:
XS GIS Cut Line= 3
      3704048.62     10208237.38      3703336.82     10207673.14
       3702307.7     10207000.78
#Sta/Elev= 30
  4095.3  307.96  4285.9  305.61  4612.8  297.09  4627.2  297.81  4662.5  295.78
  4811.4  295.48  4925.7  293.28  4947.7  294.26  4976.6  292.36    4983  288.24
    4996  288.24 5000.57292.4992  5012.4  295.81  5054.6  295.31  5075.7  291.24
  5105.9  295.51    5127  293.84  5169.6  295.19  5286.9  295.08  5380.4  291.82
  5401.5  293.59  5458.8   294.3  5546.3  293.99  5603.6  291.74  5618.7  293.34
  5691.1  293.95  6117.2  293.64  6146.6  294.59  6196.9   293.4  6232.9  303.19
#Mann= 5 ,-1 , 0
  4095.3     .17       0  4811.4     .15       0  4976.6     .09       0
 5000.57     .15       0  6117.2     .11       0
Bank Sta=4976.6,5000.57
XS Rating Curve= 0 ,0
Exp/Cntr=0.3,0.1

Type RM Length L Ch R = 1 ,325000  ,500,500,500
BEGIN DESCRIPTION:
LAKE CREEK 628.0
END DESCRIPTION:
XS GIS Cut Line= 3
      3704067.82     10207661.04      3703568.88     10207183.13
      3701982.72      10206588.1
#Sta/Elev= 30
  4309.1  305.07  4868.7  293.72  4973.7  294.13  4981.4  288.58  4994.4  288.58
 5011.25294.1615  5189.5  294.37  5236.1  289.17    5250  291.39  5274.9  290.92
  5280.2  293.01  5310.8  295.06  5330.1  291.59  5335.4  294.18  5365.7  294.77
  5513.8  291.18  5556.1   293.2  5621.9  290.47  5695.3  292.75  6058.5  293.25
  6145.3  291.67  6165.3  300.34    6176  301.95  6184.3  300.89    6208  292.76
  6229.4  291.86  6269.8  294.98  6346.8  294.73  6440.6  297.79  6694.1  313.59
#Mann= 5 ,-1 , 0
  4309.1     .17       0  4868.7     .15       0  4973.7     .09       0
 5011.25     .15       0  6145.3     .17       0
Bank Sta=4973.7,5011.25
XS Rating Curve= 0 ,0
Exp/Cntr=0.3,0.1

Type RM Length L Ch R = 1 ,324500  ,500,500,500
BEGIN DESCRIPTION:
LAKE CREEK 627.0
END DESCRIPTION:
XS GIS Cut Line= 3
      3704267.85     10207561.07      3703788.96     10206752.66
      3702767.89      10205761.1
#Sta/Elev= 30
  4060.4  306.78  4639.2  294.01  4728.7  292.46  4972.8  292.68  4994.2  288.74
  5004.3  289.44 5007.84  292.75  5129.1  293.07  5164.6  288.15    5214  293.15
  5277.8  288.84  5298.9  293.23  5348.5  293.42  5369.6  289.41  5390.9  291.72
  5397.9  288.49  5454.5  291.39  5475.6  288.34  5482.8  291.59  5503.9  292.26
  5617.1  291.44  5645.6  288.06  5772.7   291.6  6048.5  291.39  6090.9  301.16
  6119.2  293.35  6204.7   296.6  6352.7  302.06    6381  307.48  6423.3  306.08
#Mann= 6 ,-1 , 0
  4060.4     .17       0  4639.2     .11       0  4728.7     .15       0
  4972.8     .09       0 5007.84     .15       0  6204.7     .11       0
Bank Sta=4972.8,5007.84
XS Rating Curve= 0 ,0
Exp/Cntr=0.3,0.1

Type RM Length L Ch R = 1 ,324000  ,492,492,492
BEGIN DESCRIPTION:
LAKE CREEK 626.0
END DESCRIPTION:
XS GIS Cut Line= 3
      3704467.86      10207311.1      3704108.89     10206378.83
      3703117.82     10205361.04
#Sta/Elev= 30
    4001  303.46  4036.1  303.32    4082  302.65    4143  301.48  4311.8  299.55
    4494  292.84  4597.6  294.13  4690.8  291.86  4756.3  291.92  4865.7  291.24
  4990.6  292.71  4996.1  288.43    5000  288.43  5006.3  290.17  5013.2  288.68
  5020.4   293.1  5146.5  291.09  5265.1  291.03  5692.2  291.82  5720.5   290.6
  5734.6  287.49  5777.1  290.98  5953.8  289.87  6089.4  293.41  6116.4  295.51
  6137.7  301.13  6180.2  297.42    6272  304.67  6364.1  304.25  6420.6  316.04
#Mann= 12 ,-1 , 0
    4001     .17       0  4036.1     .11       0    4082     .17       0
    4143     .11       0  4690.8     .15       0  4756.3     .11       0
  4865.7     .15       0  4990.6     .09       0  5020.4     .15       0
  5146.5     .17       0  5265.1     .15       0  6089.4     .11       0
Bank Sta=4990.6,5020.4
XS Rating Curve= 0 ,0
Exp/Cntr=0.3,0.1

Type RM Length L Ch R = 1 ,323508  ,508,508,508
BEGIN DESCRIPTION:
LAKE CREEK 625.0
END DESCRIPTION:
XS GIS Cut Line= 3
      3704977.44     10207100.22      3704413.21     10206067.24
      3703317.88     10205161.09
#Sta/Elev= 30
  3712.6  303.75  3801.4   302.6  3985.1  296.73  4248.3  293.52  4552.9  293.98
  4681.5   295.9  4948.1  290.94  4983.3   291.5  4997.6  288.93  5011.9  291.74
  5090.1  290.15  5316.7  290.25    5374  288.31  5650.2  291.21  5671.8   287.7
  5685.8   287.7    5701  290.17  5750.5  291.46  5792.1  289.74  5948.4  291.24
  6022.5  297.76  6069.6  299.41  6083.9  302.38  6104.8  300.08  6133.4  302.36
  6197.2  301.49  6225.9  304.48  6261.1  301.45  6283.2   305.1  6311.2  306.18
#Mann= 5 ,-1 , 0
  3712.6     .11       0  4681.5     .15       0  4983.3     .09       0
  5011.9     .15       0  6022.5     .11       0
Bank Sta=4983.3,5011.9
XS Rating Curve= 0 ,0
Exp/Cntr=0.3,0.1

Type RM Length L Ch R = 1 ,323000  ,500,500,500
BEGIN DESCRIPTION:
LAKE CREEK 624.0
END DESCRIPTION:
XS GIS Cut Line= 3
      3705517.88     10207511.11      3704382.79     10205605.22
      3703517.88      10204611.1
#Sta/Elev= 30
  2781.7  311.58  3305.5  299.51  3517.7  302.09  4015.5  292.88  4399.7   293.3
  4527.2  290.62  4983.9  289.79  5020.3  287.41  5027.9  290.27  5204.5  288.56
  5481.7  291.05  5531.1  290.03  5538.3  286.54  5594.7  287.26    5609  290.74
  5729.5  290.14  5793.2  293.39  5835.9  290.76  5853.5  292.78    5909  297.53
  5920.4  301.68  5934.6  303.25  5970.7  293.66  5991.6  291.67  6034.3  301.91
  6062.8  301.27  6083.7  298.06  6154.9  303.35  6247.5  306.36  6317.7  309.46
#Mann= 7 ,-1 , 0
  2781.7     .11       0  4527.2     .15       0  4983.9     .09       0
  5027.9     .15       0  5853.5     .17       0    5909     .11       0
  6247.5     .15       0
Bank Sta=4983.9,5027.9
XS Rating Curve= 0 ,0
Exp/Cntr=0.3,0.1

Type RM Length L Ch R = 1 ,322500  ,500,500,500
BEGIN DESCRIPTION:
LAKE CREEK 623.0
END DESCRIPTION:
XS GIS Cut Line= 3
      3705593.76     10207143.63      3704750.44     10205354.96
      3704049.46     10204518.18
#Sta/Elev= 30
  3022.5  304.08  3478.6  295.88  3766.1  298.76    4142  291.12  4217.2  292.37
  4329.9  289.58  4887.9   288.6  4945.5  287.97  4973.8  289.08  5005.8  286.38
  5011.7  289.36  5018.2  287.65    5026  289.59  5260.2  286.76    5324  288.12
  5366.9  286.76  5395.5   288.8  5558.2  290.65  5579.1  288.61  5586.2  285.66
  5600.4  285.66  5621.9  290.06  5800.2  288.29  5870.4  289.85  5899.1  292.36
  5956.3  293.68  5968.6  295.13  6055.2  297.23  6069.5  299.07  6091.6  305.67
#Mann= 5 ,-1 , 0
  3022.5     .11       0  4887.9     .15       0  4973.8     .09       0
  5011.7     .15       0  5968.6     .11       0
Bank Sta=4973.8,5011.7
XS Rating Curve= 0 ,0
Exp/Cntr=0.3,0.1

Type RM Length L Ch R = 1 ,322000  ,500,500,500
BEGIN DESCRIPTION:
LAKE CREEK 622.0
END DESCRIPTION:
XS GIS Cut Line= 3
      3706717.84     10206111.06      3705094.92      10205088.7
      3704567.85     10204261.07
#Sta/Elev= 30
  3081.9  310.47    3199  307.22  3423.8  294.62  3800.6  291.59  3897.9  292.28
  4409.9  291.06  4522.2  290.54    4849  288.27  4973.1  287.99  5003.5  285.56
  5024.6  287.77  5170.2  286.94  5315.8  289.07  5342.9  288.33  5364.7  286.43
    5366  285.23  5388.4  285.68  5394.6  289.08  5409.8   288.8  5415.7  287.02
    5424  288.64  5509.7  289.15  5640.1  287.74  5661.2  288.57  5684.7  287.03
  5706.9   289.6  5772.3  293.05  5837.3  296.76  5900.8  303.85  5981.2  309.83
#Mann= 9 ,-1 , 0
  3081.9     .11       0  3897.9     .15       0  4409.9     .17       0
  4522.2     .11       0    4849     .15       0  4973.1     .09       0
  5024.6     .15       0  5684.7     .17       0  5772.3     .11       0
Bank Sta=4973.1,5024.6
XS Rating Curve= 0 ,0
Exp/Cntr=0.3,0.1

Type RM Length L Ch R = 1 ,321500  ,500,500,500
BEGIN DESCRIPTION:
LAKE CREEK 621.0
END DESCRIPTION:
XS GIS Cut Line= 3
      3706717.82     10206061.04      3705107.51     10204619.62
      3704617.85     10204261.07
#Sta/Elev= 30
  2838.8  310.42    2881  310.26  3129.2  295.85    3186  294.02  3284.7  294.84
  3525.5  291.18  3692.9  291.44  3886.6  290.21  4189.9  290.24  4524.3  288.71
  4609.6  287.28  4739.2  288.46  4793.5     289  4892.2  286.91  4977.4  287.04
  4989.5  283.58  5003.3  283.58  5005.9  285.22  5012.1  285.06 5018.01287.0554
  5035.2   288.3  5156.4  288.52  5242.1  288.38  5256.8  286.98  5277.6   288.1
  5321.6  287.51  5334.2  288.92  5360.2  289.35    5421  292.82  5606.9  307.18
#Mann= 7 ,-1 , 0
  2838.8     .11       0  3692.9     .15       0  4189.9     .11       0
  4739.2     .15       0  4977.4     .09       0 5018.01     .15       0
  5360.2     .11       0
Bank Sta=4977.4,5018.01
XS Rating Curve= 0 ,0
Exp/Cntr=0.3,0.1

Type RM Length L Ch R = 1 ,321000  ,500,500,500
BEGIN DESCRIPTION:
LAKE CREEK 620.0
END DESCRIPTION:
XS GIS Cut Line= 3
      3707317.82     10206011.04      3705426.05     10204275.16
      3704717.89     10204011.09
#Sta/Elev= 30
  2432.5  316.88    2963  305.14    3013  302.01  3048.1  302.39  3147.4  299.68
  3253.5  301.57  3288.6  300.85    3473  291.47  3536.5  291.83    3558  290.15
  3727.6  290.89  3770.2  296.91  3814.9   293.2  3989.7  288.42  4152.4  289.63
  4472.8  288.13  4746.8  288.16  4821.5  286.24  4846.1  285.15  4881.3   287.1
  4980.5  286.72  4987.3  286.12  4992.4  282.68  5019.4  283.48  5025.4  284.21
  5030.7  286.96  5497.6  288.56  5617.1  295.58    5680  302.98  5755.8  308.14
#Mann= 7 ,-1 , 0
  2432.5     .11       0  3814.9     .15       0  4472.8     .17       0
  4821.5     .15       0  4980.5     .09       0  5030.7     .15       0
  5497.6     .11       0
Bank Sta=4980.5,5030.7
XS Rating Curve= 0 ,0
Exp/Cntr=0.3,0.1

Type RM Length L Ch R = 1 ,320500  ,608,608,608
BEGIN DESCRIPTION:
LAKE CREEK 619.0
END DESCRIPTION:
XS GIS Cut Line= 3
      3707000.01      10205147.1      3705846.14     10204097.25
      3704867.88     10203411.09
#Sta/Elev= 30
    3440  301.45  3807.1  295.22    4026  299.03  4146.3  295.74  4259.4  289.88
  4330.8  287.15  4479.4  287.79  4656.5  285.07  4790.9   287.8    4968  283.76
  4982.1  284.59  5003.2  281.72  5017.1  281.72  5017.8  283.25    5024  284.69
  5083.2  290.43  5181.7  289.48  5195.5  290.49  5237.8  290.69  5376.7  292.31
  5425.8  290.82  5440.6  289.04  5613.1  288.09  5678.5  288.99  5684.6  290.31
  5714.3  288.76  5785.7  288.62  5943.5  292.85  6122.2  304.21  6194.9  307.07
#Mann= 7 ,-1 , 0
    3440     .11       0  4259.4     .15       0  4982.1     .09       0
    5024     .15       0  5195.5     .11       0  5237.8     .15       0
  5376.7     .11       0
Bank Sta=4982.1,5024
XS Rating Curve= 0 ,0
Exp/Cntr=0.3,0.1

Type RM Length L Ch R = 1 ,319892  ,392,392,392
BEGIN DESCRIPTION:
LAKE CREEK 618.0
END DESCRIPTION:
XS GIS Cut Line= 3
       3707321.2     10205086.35      3706322.93      10203940.5
        3704908.     10203263.42
#Sta/Elev= 30
  3634.6  305.46  3846.2  298.09  4073.1  296.17  4108.2  297.65  4264.9  296.59
  4349.4  295.21  4490.8  289.55  4597.2  290.12  4739.6  287.19  4924.5  286.18
  4944.6  286.13  4994.7  281.56  5008.6  281.56  5015.9  283.06  5022.5  282.28
  5044.3  286.38  5210.4  286.18  5234.1  283.18  5238.7  283.74  5261.2  286.41
    5293  287.75  5347.1  287.46  5592.3  287.38  5758.6  292.46  6035.7  289.36
    6366  292.76  6694.5  305.75  6711.6  310.56  6717.1  310.67  6722.9  308.68
#Mann= 7 ,-1 , 0
  3634.6     .11       0  4924.5     .15       0  4944.6     .09       0
  5044.3     .15       0  5234.1     .11       0  5238.7     .15       0
  5347.1     .11       0
Bank Sta=4944.6,5044.3
XS Rating Curve= 0 ,0
Exp/Cntr=0.3,0.1

Type RM Length L Ch R = 1 ,319500  ,590,590,590
BEGIN DESCRIPTION:
LAKE CREEK 617.0
END DESCRIPTION:
XS GIS Cut Line= 3
      3707667.82     10204861.04      3706723.44     10203911.37
      3704717.82     10203111.06
#Sta/Elev= 30
  3660.7  309.27  3851.6  305.17  3968.2  298.88  4558.7  287.67  4862.7  284.56
  4926.4  284.59  4961.7  287.44 4966.24285.8477  4983.1  280.61  5037.1     286
  5200.9  286.59  5436.7  287.49  5449.4  283.45    5467     283  5473.7   283.2
  5479.8  287.25  5522.2  287.79  5544.4  285.69  5557.2   281.2  5587.4  286.96
  5611.2  286.82  5813.5  286.77  6050.4  291.39  6545.7  293.82  6857.9  303.48
  6899.3  310.53    6929  305.95  7007.1  311.37  7042.1   309.6  7159.4  312.29
#Mann= 7 ,-1 , 0
  3660.7     .17       0  3968.2     .11       0 4966.24     .06       0
  5037.1     .15       0  5200.9     .11       0    5467     .15       0
  5611.2     .11       0
Bank Sta=4966.24,5037.1
XS Rating Curve= 0 ,0
Exp/Cntr=0.3,0.1

Type RM Length L Ch R = 1 ,318910  ,410,410,410
BEGIN DESCRIPTION:
LAKE CREEK 616.0
END DESCRIPTION:
XS GIS Cut Line= 3
      3708017.83     10204561.04      3707086.82     10203489.11
       3705067.9     10203111.08
#Sta/Elev= 30
  3686.1  311.73  3877.4  303.05  4012.3  299.77  4210.7  291.84  4607.6  286.66
  4948.1  286.18  4976.1  285.66  4983.7  284.46  4990.4  280.43  5004.3  280.43
  5018.8  285.94  5053.9  287.04  5090.1  285.43  5178.9  288.38  5241.1  285.23
  5289.2  282.23  5341.8  287.05  5376.4  286.63    5522  286.67  5557.3   285.4
  5639.9   286.5  5684.7  285.13    5939  286.23  6038.7  287.04    6112  288.86
  6208.9  288.36  6755.3  293.28  7007.3  298.67  7128.6  303.74  7159.9  302.37
#Mann= 9 ,-1 , 0
  3686.1     .11       0  4948.1     .15       0  4976.1     .09       0
  5018.8     .15       0  5241.1     .17       0  5376.4     .15       0
  5639.9     .11       0    5939     .17       0  6038.7     .11       0
Bank Sta=4976.1,5018.8
XS Rating Curve= 0 ,0
Exp/Cntr=0.3,0.1

Type RM Length L Ch R = 1 ,318500  ,500,500,500
BEGIN DESCRIPTION:
LAKE CREEK 615.0
END DESCRIPTION:
XS GIS Cut Line= 3
      3708267.85     10204211.07      3707338.11     10203247.49
      3705317.84     10202761.07
#Sta/Elev= 30
    3661  320.72    3859  307.25  4255.1  291.42  4276.2  289.79  4389.4   289.1
  4537.9  285.76  4882.6  285.61  4969.3  286.22  4983.4  284.18  4989.6   278.7
  5003.5   278.7  5005.7   281.5  5010.9  284.45  5031.1  285.53  5094.7   284.8
  5173.5  286.45  5298.6  284.93  5319.1  283.68  5339.7  285.57    5422  286.46
  5561.1  284.71  5915.7  285.06  6030.6  288.27  6158.5  288.18  6265.4  291.29
  6399.1  289.63  6666.6  292.65  6839.7  296.52  6851.7  295.59    7078  298.62
#Mann= 5 ,-1 , 0
    3661     .11       0  4882.6     .15       0  4983.4     .09       0
  5010.9     .15       0  6030.6     .11       0
Bank Sta=4983.4,5010.9
XS Rating Curve= 0 ,0
Exp/Cntr=0.3,0.1

Type RM Length L Ch R = 1 ,318000  ,472,472,472
BEGIN DESCRIPTION:
LAKE CREEK 614.0
END DESCRIPTION:
XS GIS Cut Line= 3
      3708317.86     10203661.08      3707375.06     10202839.73
      3705441.41     10202523.12
#Sta/Elev= 30
  3749.6  313.06  4259.9  287.89  4415.6  284.49    4796  285.31    4983  284.82
  5000.4  278.09  5014.3  278.09  5022.6  285.11  5037.7  286.62  5311.3  284.78
  5341.7  283.14  5390.6  285.44  5896.6  284.65    5996  285.15  6194.8  289.65
  6294.2  288.03  6375.3  290.37  6476.6  289.94  6517.1  290.86  6547.5  295.65
  6571.3  294.35  6588.1  289.59  6598.2  288.77  6679.3  287.92  6719.8  293.32
  6791.2  296.46  6851.5  299.89  6912.3  301.43  6932.6  300.38  6959.4  306.55
#Mann= 8 ,-1 , 0
  3749.6     .11       0    4796     .15       0    4983     .09       0
  5022.6     .15       0  5896.6     .17       0    5996     .11       0
  6194.8     .17       0  6791.2     .11       0
Bank Sta=4983,5022.6
XS Rating Curve= 0 ,0
Exp/Cntr=0.3,0.1
