--- LANDRUM CREEK.prj (project) ---

Proj Title=LANDRUM CREEK Base Level Engineering
Current Plan=p01
Default Exp/Contr=0.3,0.1
English Units
Geom File=g01
Flow File=f01
Plan File=p01
Y Axis Title=Elevation
X Axis Title(PF)=Main Channel Distance
X Axis Title(XS)=Station
BEGIN DESCRIPTION:
LANDRUM CREEK
END DESCRIPTION:
DSS Export Rating Curves= 0
DSS Export Rating Curve Sorted= 0
DSS Export Volume Flow Curves= 0
DXF OffsetX= 0
DXF OffsetY= 0
DXF ScaleX= 1
DXF ScaleY= 10

--- LANDRUM CREEK.p01 (plan) ---

Plan Title=Multiple Run
Short Identifier=Multiple
Geom File=g01
Flow File=f01
Subcritical Flow
K Sum by GR= 0
Std Step Tol= 0.01
Critical Tol= 0.01
Num of Std Step Trials= 20
Max Error Tol= 0.3
Flow Tol Ratio= 0.001
Split Flow NTrial= 30
Split Flow Tol= 0.02
Split Flow Ratio= 0.02
Log Output Level= 0
Friction Slope Method= 1
Unsteady Friction Slope Method= 2
Unsteady Bridges Friction Slope Method= 1
Parabolic Critical Depth
Global Vel Dist=  1 , 1 , 1
Global Log Level= 0
CheckData=True
Encroach Param= -1, 0, 0, 0
BEGIN DESCRIPTION:
Multiple Run
END DESCRIPTION:

--- LANDRUM CREEK.f01 (steady flow) ---

Flow Title=Multiple
Program Version=4.10
Number of Profiles= 7
Profile Names=10-year,25-year,50-year,1pct_min,100-year,1pct_plu,500-year
River Rch & RM=LANDRUM CREEK,Reach-1         ,38018
     493     660     884     391    1180    3564    2174
River Rch & RM=LANDRUM CREEK,Reach-1         ,33802
     595     801    1078     477    1440    4349    2663
River Rch & RM=LANDRUM CREEK,Reach-1         ,28833
    1502    2112    2927    1329    4014   12122    7814
River Rch & RM=LANDRUM CREEK,Reach-1         ,20669
    2099    2989    4176    1909    5766   17413   11388
River Rch & RM=LANDRUM CREEK,Reach-1         ,12323
    2486    3549    4963    2271    6858   20711   13554
River Rch & RM=LANDRUM CREEK,Reach-1         ,10365
    2486    3549    4963    2271    6858   20711   13554
River Rch & RM=LANDRUM CREEK,Reach-1         ,4171
    2973    4264    5981    2742    8282   25011   16448
Boundary for River Rch & Prof#=LANDRUM CREEK,Reach-1         , 1
Up Type= 0
Dn Type= 3
Dn Slope=0.002
Boundary for River Rch & Prof#=LANDRUM CREEK,Reach-1         , 2
Up Type= 0
Dn Type= 3
Dn Slope=0.002
Boundary for River Rch & Prof#=LANDRUM CREEK,Reach-1         , 3
Up Type= 0
Dn Type= 3
Dn Slope=0.002
Boundary for River Rch & Prof#=LANDRUM CREEK,Reach-1         , 4
Up Type= 0
Dn Type= 3
Dn Slope=0.002
Boundary for River Rch & Prof#=LANDRUM CREEK,Reach-1         , 5
Up Type= 0
Dn Type= 3
Dn Slope=0.002
Boundary for River Rch & Prof#=LANDRUM CREEK,Reach-1         , 6
Up Type= 0
Dn Type= 3
Dn Slope=0.002
Boundary for River Rch & Prof#=LANDRUM CREEK,Reach-1         , 7
Up Type= 0
Dn Type= 3
Dn Slope=0.002
DSS Import GetInterval= 0
DSS Import GetPeak= 0
DSS Import FillOption= 0

--- LANDRUM CREEK.g01 (geometry) ---

Geom Title=Existing Conditions
Program Version=4.10

River Reach=LANDRUM CREEK   ,Reach-1
Reach XY= 30
      3749439.03     10132986.21      3750042.33     10131195.85
      3749088.23     10129686.84      3749478.23     10129476.84
      3749678.23     10128416.84      3750208.23     10128106.84
      3750998.59     10126609.21      3750202.24     10125850.04
      3750086.36     10124757.39      3749419.91     10124045.14
      3749417.49     10121519.99      3749010.05     10120730.54
      3748495.81     10120512.43      3748629.13     10119789.51
      3748237.38     10119277.49      3748786.31     10118646.04
      3748559.13     10118060.04      3749706.63     10115795.23
      3750063.89     10113601.23      3749662.84     10112219.28
       3749737.5     10111075.19      3749027.43     10109526.57
      3749438.89     10108892.89      3748975.51     10108355.32
      3749305.91     10108386.99       3749236.3     10107738.28
      3748802.91     10107418.05      3748671.71     10107719.15
      3748541.52     10106780.86      3747978.23     10106906.84

Type RM Length L Ch R = 1 ,38018   ,405,405,405
BEGIN DESCRIPTION:
LANDRUM CREEK 65.0
END DESCRIPTION:
XS GIS Cut Line= 3
        3749819.     10132878.35       3749346.8     10132817.59
      3748970.06     10133037.07
#Sta/Elev= 30
  4527.5  309.01  4538.7  309.06  4629.5  304.02  4703.6  301.68  4794.1  297.83
  4857.6  296.87  4891.6  297.48  4937.1  296.92  4952.1  297.33  4972.3  296.58
  4998.5  294.51  4998.8  294.01  5013.9  294.94  5020.1  296.45  5041.6  299.32
  5063.1  299.17  5073.1  299.81  5106.8  300.85  5121.8  300.71  5152.8   302.3
  5230.1  303.77  5268.6  305.45  5282.3  305.06  5313.7  306.35  5326.4  305.97
  5340.4  306.89  5362.5   307.4  5378.3  308.78    5394  307.99  5439.6  309.24
#Mann= 8 ,-1 , 0
  4527.5     .11       0  4794.1     .17       0  4972.3     .09       0
  5020.1     .17       0  5073.1     .15       0  5106.8     .17       0
  5230.1     .11       0  5340.4     .17       0
Bank Sta=4972.3,5020.1
XS Rating Curve= 0 ,0
Exp/Cntr=0.3,0.1

Type RM Length L Ch R = 1 ,37613   ,661,661,661
BEGIN DESCRIPTION:
Mapping XS 3b483a20
END DESCRIPTION:
XS GIS Cut Line= 3
      3749869.41     10132591.91      3749480.48     10132453.01
       3749072.7     10132732.38
#Sta/Elev= 30
  4618.7  303.64  4636.2  303.85  4661.7   301.2  4723.2  299.84  4832.7  295.84
  4929.3  293.07  4949.5  293.21  4964.3   292.2  4981.4  292.47  5000.6  291.72
  5000.9  291.22  5004.4  291.22  5004.6  291.72  5013.2   292.5  5068.8  292.72
  5083.4  293.27  5137.3  292.95  5176.5   293.7  5182.5  294.54    5241  294.78
  5269.2  296.43  5284.1  295.52  5313.7  296.02  5370.8   298.7  5391.7  298.77
  5421.5  299.73  5463.5  299.29  5499.4  300.58  5514.3  300.44    5526  301.29
#Mann= 5 ,-1 , 0
  4618.7     .11       0  4929.3     .15       0  4981.4     .09       0
  5013.2     .15       0  5137.3     .17       0
Bank Sta=4981.4,5013.2
XS Rating Curve= 0 ,0
Exp/Cntr=0.3,0.1

Type RM Length L Ch R = 1 ,36952   ,500,500,500
BEGIN DESCRIPTION:
Mapping XS 90754568
END DESCRIPTION:
XS GIS Cut Line= 3
      3750133.28     10132361.02      3749886.73     10131935.65
      3749342.21     10132025.82
#Sta/Elev= 30
  4568.6  300.74    4668  296.99    4711  296.04  4769.8  293.42  4822.8  292.21
  4887.5  289.23  4961.5  287.92  4967.8  286.92  4973.6  287.03  4983.5  285.38
  5003.1  284.33  5003.3  283.83  5010.9  284.73  5026.6  285.15  5048.1  286.94
    5060  286.55    5162  287.41  5190.9  288.23    5201  287.19  5211.2  288.02
  5231.4  287.85  5264.9  288.93  5353.1  290.06  5383.5  289.59  5413.9  290.53
  5454.4  292.76  5474.7  292.04  5565.9  294.35  5576.1  295.18  5612.2  295.37
#Mann= 5 ,-1 , 0
  4568.6     .11       0  4983.5     .09       0  5026.6     .15       0
    5162     .11       0  5264.9     .15       0
Bank Sta=4983.5,5026.6
XS Rating Curve= 0 ,0
Exp/Cntr=0.3,0.1

Type RM Length L Ch R = 1 ,36452   ,274,274,274
BEGIN DESCRIPTION:
Mapping XS 38d6506c
END DESCRIPTION:
XS GIS Cut Line= 3
      3750463.16     10131647.46      3749777.36     10131458.21
      3749419.29     10131847.42
#Sta/Elev= 30
  4574.2  292.88  4621.7  290.84  4650.9  290.56  4690.4  288.73  4797.6   285.6
  4803.9   284.5  4826.7  283.44  4826.9  282.94  4830.4  282.94  4830.7  283.44
  4877.8  284.03  4917.3  283.65  5150.3  284.16  5160.6  284.62  5386.2  283.68
  5414.5  285.35  5421.9  285.84  5563.1  288.15  5641.4  289.21  5683.6   289.1
  5690.7  289.79  5697.5  289.31  5702.7   289.7  5711.7  290.33  5719.1   289.9
  5768.4  291.26  5782.6  290.56    5790  290.71  5796.8  290.96  5814.5   292.9
#Mann= 4 ,-1 , 0
  4574.2     .11       0  4797.6     .07       0  5414.5     .11       0
  5702.7     .15       0
Bank Sta=4797.6,5414.5
XS Rating Curve= 0 ,0
Exp/Cntr=0.3,0.1

Type RM Length L Ch R = 1 ,36178   ,144,144,144
BEGIN DESCRIPTION:
Mapping XS 2895d314
END DESCRIPTION:
XS GIS Cut Line= 3
      3750466.63     10131633.59      3749938.82     10131171.76
      3749294.72     10131121.41
#Sta/Elev= 30
  4438.8  292.66  4496.4   291.3  4510.6  290.43  4517.3  290.64  4524.8  290.07
  4659.6  286.09  4702.3   284.9  4723.2  283.38  4772.6  283.45    4801  284.18
    4858  283.61  4876.9   283.1  4877.1   282.6  4880.6   282.6  4880.9   283.1
  4907.3  284.04  4950.1  284.53  4999.4     284  5027.9  284.42  5214.7  283.73
  5391.9  283.94  5452.1  286.05  5502.2  287.68  5532.3  289.65  5542.3  289.49
  5612.5  291.85  5692.8  292.17  5732.9  292.98    5753  292.84  5786.2  293.72
#Mann= 3 , 0 , 0
  4438.8     .11       0  4659.6     .06       0  5452.1     .11       0
Bank Sta=4659.6,5452.1
XS Rating Curve= 0 ,0
Exp/Cntr=0.3,0.1

Type RM Length L Ch R = 1 ,36034   ,141,141,141
BEGIN DESCRIPTION:
Mapping XS b98e2b37
END DESCRIPTION:
XS GIS Cut Line= 6
      3750468.35     10131616.23      3750225.28     10131345.37
      3750112.43     10131192.59      3749983.96      10131091.9
      3749867.64     10131031.13      3749296.46     10131102.31
#Sta/Elev= 30
    4335  292.55  4572.4  285.51  4657.7  286.91  4800.8  286.73  4821.6  287.35
  4836.2   286.6  4857.1  287.41  4886.4   286.6  4893.7  287.21  4900.2  286.53
  4907.6   287.3  4928.6  286.93    4957  287.61  4977.8  286.93  4986.6  287.48
  4992.7  286.79  5127.1  287.25    5132  286.61  5169.9  287.31  5175.6  286.69
  5203.6   287.4  5334.5   287.6  5399.5  286.97 5403.73  286.31  5425.9  284.16
  5447.8  286.37  5558.3  290.75  5628.7  291.86    5696  291.94  5760.7  293.47
#Mann= 3 , 0 , 0
    4335     .11       0 5403.73     .06       0  5447.8     .11       0
Bank Sta=5403.73,5447.8
XS Rating Curve= 0 ,0
Exp/Cntr=0.3,0.1

Type RM Length L Ch R = 1 ,35893   ,486,486,486
BEGIN DESCRIPTION:
Mapping XS 7f96e4a9
END DESCRIPTION:
XS GIS Cut Line= 5
       3750596.8     10131482.52      3750081.18     10131022.45
       3749846.8     10130930.44      3749565.55      10130928.7
      3749302.87     10131066.05
#Sta/Elev= 30
    4211  294.11  4359.8  289.21  4409.9   288.4  4445.1  286.16  4487.7   286.2
  4516.1  284.55  4608.1  283.37  4714.3  279.69  4735.2  280.36  4777.8  278.03
  4827.1  278.96  4915.2  277.15  4950.4  277.23  4999.3  274.62  5002.9  273.62
  5023.7  275.69    5029  275.19  5150.6  277.33  5192.8  278.33  5232.8  280.57
  5312.8  281.96  5342.8  284.26  5352.8  284.34  5362.8  282.74  5372.8  282.24
  5392.8  283.73  5522.8  289.42  5703.3  291.76  5725.9  293.85  5731.5  295.54
#Mann= 3 , 0 , 0
    4211     .11       0  4950.4     .06       0  5150.6     .11       0
Bank Sta=4950.4,5150.6
XS Rating Curve= 0 ,0
Exp/Cntr=0.3,0.1

Type RM Length L Ch R = 1 ,35407   ,483,483,483
BEGIN DESCRIPTION:
Mapping XS 24622606
END DESCRIPTION:
XS GIS Cut Line= 3
      3750240.94     10130538.07      3749753.05     10130562.38
      3749287.76     10131032.88
#Sta/Elev= 30
  4511.7  290.87  4524.8  290.83  4604.9  286.53  4634.9  285.99  4676.2  282.71
    4705  282.14  4735.1  279.48  4785.1  277.66  4865.2  273.24  4945.3  273.32
  4983.4   272.6  4983.6   272.1  5017.1  273.56  5024.2  273.15  5031.2  274.28
  5038.3  273.53  5045.4  274.49  5066.6  273.98  5200.9  277.96  5236.3   279.8
  5335.3  282.98  5420.2  287.24  5476.7  288.54  5483.8  289.33  5582.8  290.62
  5611.1  290.78  5618.1  290.18  5646.4  291.56  5658.3  294.16  5661.9  294.16
#Mann= 3 , 0 , 0
  4511.7     .11       0  4785.1     .06       0  5200.9     .11       0
Bank Sta=4785.1,5200.9
XS Rating Curve= 0 ,0
Exp/Cntr=0.3,0.1

Type RM Length L Ch R = 1 ,34924   ,416,416,416
BEGIN DESCRIPTION:
LANDRUM CREEK 64.0
END DESCRIPTION:
XS GIS Cut Line= 3
      3750067.88     10130061.07      3749476.35     10130167.94
      3749003.36     10130572.65
#Sta/Elev= 30
  4398.9   289.8    4583  280.51  4632.6  278.31    4655  278.24  4693.6  275.29
  4703.5  273.91  4708.6  274.22  4713.9  273.62  5050.7  273.13    5058  273.43
  5072.2   276.1  5086.5  275.57  5107.3  272.71  5135.9  273.12  5150.2  272.69
  5154.7  272.34    5155  271.84    5171  273.23    5193  272.78  5199.6  273.49
  5207.2  272.87  5213.8  274.47  5221.5  273.43  5228.1  275.32  5363.1  278.28
  5511.3  282.28  5582.7  284.86  5590.3  285.45  5611.2  290.04  5622.5  290.37
#Mann= 4 ,-1 , 0
  4398.9     .11       0    4583     .15       0    4655     .06       0
  5363.1     .11       0
Bank Sta=4655,5363.1
XS Rating Curve= 0 ,0
Exp/Cntr=0.3,0.1

Type RM Length L Ch R = 1 ,34508   ,180,180,180
BEGIN DESCRIPTION:
LANDRUM CREEK 63.0
END DESCRIPTION:
XS GIS Cut Line= 3
       3750168.7     10129687.26      3749227.62     10129836.23
      3748916.53     10129965.04
#Sta/Elev= 30
  4047.2  294.78  4071.6  294.17  4103.6  293.68  4118.9  291.88  4139.2  291.55
    4166  289.04  4171.1  289.65  4228.4   286.5  4270.8  285.19  4311.3  281.92
  4351.8  279.78  4358.1  278.68  4382.2  278.19  4402.4     277  4420.5  274.28
  4425.5  274.94  4432.8  273.79  4487.9  273.66  4522.2  272.28    4534     273
  4645.4   273.5  4918.8  273.22  4959.3  276.55  5026.3  275.93  5097.2  278.39
  5156.6   281.1  5180.4  282.97    5263  285.41  5286.8  287.22  5336.7  288.86
#Mann= 4 ,-1 , 0
  4047.2     .17       0  4071.6     .11       0  4382.2     .06       0
  5097.2     .11       0
Bank Sta=4382.2,5097.2
XS Rating Curve= 0 ,0
Exp/Cntr=0.3,0.1

Type RM Length L Ch R = 1 ,34328   ,526,526,526
BEGIN DESCRIPTION:
LANDRUM CREEK 62.0
END DESCRIPTION:
XS GIS Cut Line= 4
        3750186.      10129626.5      3749563.22     10129617.82
      3749090.13     10129711.13      3748867.86     10129911.06
#Sta/Elev= 30
  3905.5  294.95  3923.7  294.91  3937.4  293.94  3973.7   292.9  3993.7  290.93
  4033.7  290.28  4066.8  287.66  4133.7  284.17  4153.7  282.58  4203.7  280.34
  4383.7   281.1  4463.7  282.86  4511.3   282.9  4584.8  282.94  4621.6  282.26
  4635.7  282.72  4713.5  281.74  4826.8  280.94  4921.1  281.29  4961.9   280.7
  4985.9  279.46  5007.2  278.31  5007.4  277.81  5040.5  279.32  5104.3  283.45
  5167.9  285.33  5238.9  288.69  5259.8  288.77  5267.3  289.56  5309.5  290.57
#Mann= 6 ,-1 , 0
  3905.5     .17       0  4066.8     .11       0  4511.3     .15       0
  4713.5     .11       0  4985.9     .06       0  5040.5     .11       0
Bank Sta=4985.9,5040.5
XS Rating Curve= 0 ,0
Exp/Cntr=0.3,0.1

Type RM Length L Ch R = 1 ,33802   ,333,333,333
BEGIN DESCRIPTION:
LANDRUM CREEK 61.0
END DESCRIPTION:
XS GIS Cut Line= 3
      3750034.13     10129517.99       3749469.9     10129483.27
      3748955.59     10129500.63
#Sta/Elev= 30
  4436.5   287.1  4452.8  286.91  4472.7  285.79  4492.9  283.85    4533  282.25
    4553  280.42  4623.1  276.74  4643.2  274.68  4703.3  271.05  4733.3  268.22
  4743.4  267.81  4753.4  266.57  4773.4  265.34  4843.5  264.45  4863.6  264.75
  4873.6  265.46  4903.7  265.37  4911.7  263.51  4911.9  263.01 4949.83265.3975
  5063.9     266  5093.9  267.44    5214  270.33    5294  271.74    5344   271.7
  5385.2  273.57  5424.1  273.86  5484.1  275.95  5512.8  280.09  5516.4  280.09
#Mann= 4 ,-1 , 0
  4436.5     .17       0  4472.7     .11       0  4903.7     .06       0
 4949.83     .11       0
Bank Sta=4903.7,4949.83
XS Rating Curve= 0 ,0
Exp/Cntr=0.3,0.1

Type RM Length L Ch R = 1 ,33469   ,535,535,535
BEGIN DESCRIPTION:
LANDRUM CREEK 60.0
END DESCRIPTION:
XS GIS Cut Line= 3
      3750067.89     10129361.08      3749465.56      10129190.3
      3748955.57     10129086.13
#Sta/Elev= 30
  4376.7  287.09  4432.8   284.7  4449.5  282.23  4497.5  279.98  4522.3  278.66
  4539.8  276.99  4578.9  275.28  4612.8  272.26  4771.7  264.92  4803.2  263.95
  4837.1     264  4896.5  262.63    4938  263.19  4958.8  264.24    4978  263.84
    4990  262.25    4997  261.98  4997.2  261.48  5019.8  263.99  5024.9  263.25
  5041.3  264.28  5051.5  264.05  5070.3  264.84  5143.3  265.03  5316.8  269.39
  5367.9  271.59  5373.3  272.31  5423.8  273.78  5449.5  275.79  5523.3  278.19
#Mann= 4 ,-1 , 0
  4376.7     .17       0  4497.5     .11       0    4978     .07       0
  5019.8     .11       0
Bank Sta=4978,5019.8
XS Rating Curve= 0 ,0
Exp/Cntr=0.3,0.1

Type RM Length L Ch R = 1 ,32934   ,276,276,276
BEGIN DESCRIPTION:
LANDRUM CREEK 59.0
END DESCRIPTION:
XS GIS Cut Line= 3
      3750017.86     10129011.07      3749718.23     10128916.84
      3749117.82     10128861.07
#Sta/Elev= 30
  4685.9  277.46  4759.3  273.76  4766.9  272.84  4790.7  272.25  4811.7  270.39
  4822.2  270.67  4843.2  268.42  4869.3  268.39  4874.6  267.63  4934.1   264.8
  4966.5   263.8  4971.7  263.35  4979.4  261.34 4987.27257.8247  4995.8  253.63
  5002.7  254.13  5006.6257.8538  5011.9   258.2  5020.5  261.12  5080.7  261.17
    5141  262.19    5151  261.44  5181.2  262.48  5231.4  262.23  5261.5  262.82
  5329.7  264.49  5452.3     269  5472.4  268.82  5512.6  270.06    5603  274.09
#Mann= 3 ,-1 , 0
  4685.9     .11       0 4987.27     .07       0  5006.6     .11       0
Bank Sta=4987.27,5006.6
XS Rating Curve= 0 ,0
Exp/Cntr=0.3,0.1

Type RM Length L Ch R = 1 ,32658   ,717,717,717
BEGIN DESCRIPTION:
LANDRUM CREEK 58.0
END DESCRIPTION:
XS GIS Cut Line= 3
      3749995.06     10128838.73      3749680.41     10128682.49
      3749122.77     10128608.71
#Sta/Elev= 30
  4646.5  270.48  4723.5  268.16  4745.9  266.27  4762.8  265.96  4807.6  263.11
  4835.6  262.68  4911.3   260.1    4942  260.45    4956  262.46  4964.4  262.26
    4970  260.95  4978.3  260.26 4984.45256.5119  4986.8  255.08  4992.4  253.69
  4994.7  250.32  5001.6  250.82 5009.93256.4452  5020.6  260.07  5030.6  260.08
  5040.7  259.37  5060.9  259.37  5091.2  260.65  5124.7  261.14  5212.2  263.81
  5252.6  265.57  5262.6  265.24    5303  266.24  5484.6  268.81  5560.3  271.78
#Mann= 3 ,-1 , 0
  4646.5     .11       0 4984.45     .07       0 5009.93     .11       0
Bank Sta=4984.45,5009.93
XS Rating Curve= 0 ,0
Exp/Cntr=0.3,0.1

Type RM Length L Ch R = 1 ,31941   ,568,568,568
BEGIN DESCRIPTION:
LANDRUM CREEK 57.0
END DESCRIPTION:
XS GIS Cut Line= 3
      3750167.85     10128511.07      3750018.23     10128296.84
      3749717.82     10128061.05
#Sta/Elev= 30
  4738.7     266  4760.9  265.98  4775.3  264.79  4824.1   263.6  4855.4   261.8
  4897.3  260.97  4924.9  258.69  4933.6   258.8  4946.1  257.71  4969.4  257.96
  4982.6  255.65  4987.3  254.02  4990.3  252.98    4996  249.52    5000  249.52
  5002.3  246.88  5005.8  246.88  5012.1  250.26 5019.47253.0265  5025.9  255.44
    5033  256.05  5076.3  255.28  5086.4  255.76  5103.5  256.05  5117.9  255.54
  5175.8   257.4  5254.4  258.77  5260.7  258.45  5304.1  259.64  5381.9  262.93
#Mann= 6 ,-1 , 0
  4738.7     .17       0  4855.4     .11       0  4987.3     .15       0
  4990.3     .09       0 5019.47     .15       0  5086.4     .11       0
Bank Sta=4990.3,5019.47
XS Rating Curve= 0 ,0
Exp/Cntr=0.3,0.1

Type RM Length L Ch R = 1 ,31373   ,373,373,373
BEGIN DESCRIPTION:
LANDRUM CREEK 56.0
END DESCRIPTION:
XS GIS Cut Line= 3
      3750517.89      10128111.1      3750314.09     10127929.45
      3749917.83     10127661.06
#Sta/Elev= 30
  4720.9  264.31  4770.7  263.81  4813.3   261.2  4848.5  260.09  4876.9  257.95
  4962.1  254.28  4965.4  253.55  4983.1  249.79  4988.9  247.87  4993.9  247.87
  4997.7  245.96  5001.7   244.7    5002   244.2  5012.6  244.76  5018.7  247.65
  5033.6  249.65  5069.6  251.19  5105.5     251  5130.1  252.51  5141.5  253.37
  5192.4   254.3  5198.4     254  5264.3  255.69  5270.3  255.42  5300.2   256.6
  5321.2  256.33  5342.2   256.8  5363.8  257.77    5400  260.86  5472.5  263.66
#Mann= 5 ,-1 , 0
  4720.9     .17       0  4965.4     .15       0  4983.1     .09       0
  5033.6     .15       0  5130.1     .11       0
Bank Sta=4983.1,5033.6
XS Rating Curve= 0 ,0
Exp/Cntr=0.3,0.1

Type RM Length L Ch R = 1 ,31000   ,431,431,431
BEGIN DESCRIPTION:
LANDRUM CREEK 55.0
END DESCRIPTION:
XS GIS Cut Line= 3
      3750674.37     10127836.17      3750496.38     10127669.03
      3749917.82     10127261.05
#Sta/Elev= 30
  4755.6  264.19  4806.1  262.68  4827.5  262.82    4870  260.27    4891  260.12
  4912.5  257.83  4947.7  255.62  4961.9  252.73    4976  248.72  4983.3  246.74
  4988.4  243.45  5001.9  244.46  5004.5   246.8 5014.94 248.763  5019.3  249.64
  5083.6  249.99  5105.5  246.17  5126.4  247.47  5141.2  249.97  5169.3  248.25
  5197.8  251.44  5221.3  251.22  5304.9  252.71  5328.3  252.42  5370.2  254.38
    5385  253.96  5420.7  255.04  5578.3  265.02  5628.9  269.25  5707.7  273.76
#Mann= 4 ,-1 , 0
  4755.6     .17       0    4976     .09       0 5014.94     .15       0
  5221.3     .11       0
Bank Sta=4976,5014.94
XS Rating Curve= 0 ,0
Exp/Cntr=0.3,0.1

Type RM Length L Ch R = 1 ,30569   ,586,586,586
BEGIN DESCRIPTION:
LANDRUM CREEK 54.0
END DESCRIPTION:
XS GIS Cut Line= 3
      3750745.93     10127738.45      3750544.12     10127321.81
      3749967.81     10127211.06
#Sta/Elev= 30
  4587.1  263.37  4665.3  261.35  4704.9  259.48  4710.4  258.39  4717.5   258.9
  4736.5  257.91    4750  257.29  4755.6  258.13    4762  257.98  4806.4   255.6
  4839.7  254.73  4868.5  252.67  4906.4  251.27  4941.8  248.33  4973.1   247.5
  4982.4  246.53  4986.9  246.46  5002.2  240.59  5005.7  240.59  5017.5  244.52
  5026.5  246.06  5039.7  247.13    5087  246.99  5136.9  248.47  5331.4  253.13
  5372.1  255.88    5455  259.32  5610.9  270.01  5616.5  270.93  5636.9  271.58
#Mann= 6 ,-1 , 0
  4587.1     .17       0  4736.5     .15       0  4982.4     .17       0
  4986.9     .09       0  5026.5     .17       0  5136.9     .11       0
Bank Sta=4986.9,5026.5
XS Rating Curve= 0 ,0
Exp/Cntr=0.3,0.1

Type RM Length L Ch R = 1 ,29983   ,1150,1150,1150
BEGIN DESCRIPTION:
LANDRUM CREEK 53.0
END DESCRIPTION:
XS GIS Cut Line= 3
      3751318.83     10127567.02      3750481.19     10127061.39
      3750275.22       10126966.
#Sta/Elev= 30
  4023.4  260.69  4043.3   261.9  4122.9  259.27  4138.4  259.96  4246.5  257.45
    4445  254.72  4509.1  251.77  4567.4  252.13  4625.6  248.47  4671.4  247.64
  4751.4  246.47  4757.6  245.98  4763.4  246.88  4787.3  244.58  4807.1  243.47
  4821.6   244.1  4837.2  246.19  4858.5  244.82  4888.9  245.94  4938.1  243.95
  4990.5  243.84  4996.3  241.57  4999.1  238.44  5006.4  238.94 5015.01243.9314
  5018.3  246.17  5027.5  249.24  5041.2  250.86  5058.6  250.81  5228.8  260.35
#Mann= 6 ,-1 , 0
  4023.4     .17       0  4671.4     .15       0  4751.4     .17       0
  4787.3     .15       0  4990.5     .06       0 5015.01     .11       0
Bank Sta=4990.5,5015.01
XS Rating Curve= 0 ,0
Exp/Cntr=0.3,0.1

Type RM Length L Ch R = 1 ,28833   ,511,511,511
BEGIN DESCRIPTION:
LANDRUM CREEK 52.0
END DESCRIPTION:
XS GIS Cut Line= 3
      3751675.55     10126281.44      3750967.99     10126514.64
      3750296.92     10126806.79
#Sta/Elev= 30
    4255  261.38  4266.1  260.62  4442.1  251.22  4491.5  250.07  4547.4  247.24
  4668.7  245.15  4753.6   244.6  4846.2  243.69  4872.7  242.66  4915.9  242.52
  4941.5  241.06    4958   241.6  4979.1  240.82  4989.6  236.61  4994.3  232.88
  5000.5  232.88  5004.6  235.34  5011.1  234.55    5022  240.32    5028  242.35
  5033.5  242.46  5103.8  241.47  5141.9  242.33  5150.6  241.64  5202.4  241.93
  5482.5  250.02    5506   251.4    5634  253.41  5704.3  256.63  5731.9  257.17
#Mann= 7 ,-1 , 0
    4255     .11       0  4266.1     .17       0  4668.7     .11       0
  4753.6     .15       0  4979.1     .09       0    5022     .15       0
  5202.4     .11       0
Bank Sta=4979.1,5022
XS Rating Curve= 0 ,0
Exp/Cntr=0.3,0.1

Type RM Length L Ch R = 1 ,28322   ,699,699,699
BEGIN DESCRIPTION:
LANDRUM CREEK 51.0
END DESCRIPTION:
XS GIS Cut Line= 3
      3751581.76     10126112.18       3750647.8     10126350.96
      3750303.13     10126721.55
#Sta/Elev= 30
    4036  258.62  4130.1  254.01  4145.9  253.63  4232.9  251.58  4380.6  246.43
  4438.7  245.76  4490.8  244.86  4579.2  243.68  4614.9  244.27  4620.1  243.31
  4783.4  240.34  4803.8  241.14  4819.1  239.88  4824.5  241.29  4834.8  241.74
  4859.9  239.11  4900.7  241.29  4922.6  239.34  4927.7  238.48  4941.5  240.14
  4982.4  240.89  4989.6  236.48  4994.2  231.43  5007.1  232.03 5040.44 240.886
  5049.6  242.62    5099   244.2  5106.3  245.35  5389.2  250.86  5506.1  254.83
#Mann= 9 ,-1 , 0
    4036     .11       0  4130.1     .17       0  4145.9     .11       0
  4232.9     .17       0  4438.7     .11       0  4490.8     .15       0
  4922.6     .11       0  4982.4     .06       0 5040.44     .11       0
Bank Sta=4982.4,5040.44
XS Rating Curve= 0 ,0
Exp/Cntr=0.3,0.1

Type RM Length L Ch R = 1 ,27623   ,530,530,530
BEGIN DESCRIPTION:
LANDRUM CREEK 50.0
END DESCRIPTION:
XS GIS Cut Line= 3
      3751267.82     10125561.09      3750498.42     10125903.37
      3749993.25     10126330.91
#Sta/Elev= 30
  4157.9  267.47  4234.5  265.19  4324.7  260.76  4336.2   260.3  4415.6  253.54
  4612.7  243.86  4687.8  241.47  4764.2  240.75  4773.8  240.61  4945.9  239.69
  4959.9  239.27  4983.1  236.56  4994.3  230.34  5005.7  231.06  5013.5  236.82
  5040.9  239.73  5091.5  239.97  5147.4  237.14  5169.5  238.82  5247.5  241.04
  5268.3  243.62  5282.6  243.12  5411.4   246.2  5432.1  246.45  5467.2  249.53
  5473.7  248.63  5510.1  250.42  5573.8  251.03  5607.3  252.93  5661.8  254.59
#Mann= 10 ,-1 , 0
  4157.9     .11       0  4324.7     .17       0  4336.2     .15       0
  4612.7     .17       0  4764.2     .11       0  4773.8     .15       0
  4983.1     .09       0  5013.5     .15       0  5411.4     .17       0
  5607.3     .11       0
Bank Sta=4983.1,5013.5
XS Rating Curve= 0 ,0
Exp/Cntr=0.3,0.1

Type RM Length L Ch R = 1 ,27093   ,467,467,467
BEGIN DESCRIPTION:
LANDRUM CREEK 49.0
END DESCRIPTION:
XS GIS Cut Line= 3
      3751118.24     10125416.86      3750198.04     10125809.32
      3749811.94     10125810.09
#Sta/Elev= 30
  3999.6  262.46  4048.8  259.88  4148.7  252.47  4177.7  251.84  4211.8  249.83
  4320.9  246.15  4391.4   243.6  4472.4  241.86    4630  238.79  4750.2   238.5
  4835.2  239.35  4887.9   237.4    4935  238.47    4946  237.53  4969.6  238.25
  4978.5  238.03  4987.8   234.9  4993.2  236.48  4993.6  230.17  4994.1  229.67
  5010.2  230.85  5020.2  236.09  5030.2   239.5  5090.2  243.22  5100.2  242.94
  5120.2  244.48  5210.2   246.7  5249.1  247.01  5310.2  247.26  5386.1  248.93
#Mann= 7 ,-1 , 0
  3999.6     .17       0  4211.8     .15       0  4320.9     .17       0
  4472.4     .15       0  4993.2     .09       0  5020.2     .15       0
  5249.1     .17       0
Bank Sta=4993.2,5020.2
XS Rating Curve= 0 ,0
Exp/Cntr=0.3,0.1

Type RM Length L Ch R = 1 ,26626   ,487,487,487
BEGIN DESCRIPTION:
LANDRUM CREEK 48.0
END DESCRIPTION:
XS GIS Cut Line= 3
      3750979.56      10125127.4      3750278.01     10125405.89
      3749498.42     10125752.81
#Sta/Elev= 30
  4245.2  262.03  4301.9  259.02    4355  254.56  4403.6  252.49  4666.6  242.43
  4722.5  241.27    4828  237.61    4895   236.5  4943.6  237.53  4967.9  235.97
  4973.3  233.76  4978.7  234.07  4989.4  231.98  4999.7  228.36  5006.4  228.36
  5011.1  229.92  5020.8   236.4    5044  236.11  5049.5  237.33  5065.8  237.66
  5124.7  236.02    5148  238.31  5153.5  237.68  5256.4  241.04  5350.4  242.19
  5414.6  245.09  5570.5  247.13  5755.4  251.41  5821.1  254.06  5853.3  254.03
#Mann= 6 ,-1 , 0
  4245.2     .11       0  4301.9     .17       0  4722.5     .15       0
  4967.9     .09       0  5020.8     .15       0  5256.4     .17       0
Bank Sta=4967.9,5020.8
XS Rating Curve= 0 ,0
Exp/Cntr=0.3,0.1

Type RM Length L Ch R = 1 ,26139   ,500,500,500
BEGIN DESCRIPTION:
LANDRUM CREEK 47.0
END DESCRIPTION:
XS GIS Cut Line= 3
      3750567.82     10124861.08       3750152.4     10124961.55
      3749718.46     10125464.93
#Sta/Elev= 30
  4572.6  247.73    4588  246.93  4644.6  243.21  4679.8  242.38  4721.6  239.13
  4757.8   238.1  4810.4  234.26  4829.8  234.08  4852.3  235.57  4894.1  232.11
  4922.4  235.62  4942.9  236.72 4979.83235.7026  4984.1  234.32  4994.4   228.8
  4996.4   226.5  5010.3  227.64  5016.9  235.85  5024.6  233.84  5066.3  236.58
  5109.1  235.66  5223.1  237.49  5239.7  238.78  5321.9  238.92  5393.2  242.08
  5428.3  241.42  5491.9  243.42  5563.2  243.33  5633.5  245.47  5664.6  245.49
#Mann= 5 ,-1 , 0
  4572.6     .17       0    4588     .15       0 4979.83     .09       0
  5016.9     .15       0  5239.7     .17       0
Bank Sta=4979.83,5016.9
XS Rating Curve= 0 ,0
Exp/Cntr=0.3,0.1

Type RM Length L Ch R = 1 ,25639   ,551,551,551
BEGIN DESCRIPTION:
LANDRUM CREEK 46.0
END DESCRIPTION:
XS GIS Cut Line= 3
      3750567.89     10124311.05      3749885.33     10124724.09
      3749317.84     10124761.07
#Sta/Elev= 30
  4202.2  262.08  4260.7  260.24  4369.1  253.26  4477.9  248.73  4522.3  248.06
    4565  244.68  4611.3  242.94  4681.5  236.67  4718.2  235.38  4770.6  235.36
  4813.3  232.71  4856.8  235.13  4923.8   235.4  4960.7  233.61    4982  234.41
  4987.9  232.83  4995.6   228.8    5000   228.8  5003.7  224.94  5011.2  224.94
  5031.5  233.35  5077.6  233.14  5137.8  236.93    5228  237.13  5358.2  242.89
  5414.4  244.22  5478.5  246.25  5508.6  245.32  5538.6  249.99  5568.7  250.46
#Mann= 5 ,-1 , 0
  4202.2     .11       0  4477.9     .15       0  4987.9     .09       0
  5031.5     .15       0  5414.4     .17       0
Bank Sta=4987.9,5031.5
XS Rating Curve= 0 ,0
Exp/Cntr=0.3,0.1

Type RM Length L Ch R = 1 ,25088   ,983,983,983
BEGIN DESCRIPTION:
LANDRUM CREEK 45.0
END DESCRIPTION:
XS GIS Cut Line= 3
      3750446.31     10124091.36      3749664.69      10124424.6
      3749367.85     10124561.07
#Sta/Elev= 30
  4150.3  256.97  4210.9  252.98  4392.5  246.41  4416.1   243.9  4421.6  244.14
  4539.7  236.12  4744.9  232.76  4804.8  232.84  4844.4  232.41  4887.8  234.26
  4897.5  233.07    4903   233.5  4909.6  232.47  4920.5  232.63  4979.3  229.42
  5004.5  224.75  5012.1  224.75  5018.5  228.52 5021.85229.5343  5025.7   230.7
  5040.5  231.14  5048.7  232.39  5114.8  235.39  5192.1  238.51  5215.1   237.9
  5243.5     241  5260.7  241.58  5266.5  243.49    5295   244.1  5326.7  246.94
#Mann= 5 ,-1 , 0
  4150.3     .11       0  4804.8     .15       0  4979.3     .09       0
 5021.85     .15       0  5114.8     .17       0
Bank Sta=4979.3,5021.85
XS Rating Curve= 0 ,0
Exp/Cntr=0.3,0.1

Type RM Length L Ch R = 1 ,24105   ,447,447,447
BEGIN DESCRIPTION:
LANDRUM CREEK 44.0
END DESCRIPTION:
XS GIS Cut Line= 3
      3750367.84     10123761.07      3749516.36     10123726.08
      3749204.15     10123737.18
#Sta/Elev= 30
  4147.8  255.43  4207.8   250.7  4247.9  248.97    4408  237.52    4458  234.68
  4668.2  231.59  4748.3  231.27  4798.3  231.86  4808.3  231.57  4828.4  227.71
  4838.4  226.96  4848.3  227.15  4858.4  226.37  4868.4  228.22  4878.4  231.03
  4938.5  231.09  4958.5  232.11  4978.5  231.65  4988.5  227.88  4992.9  221.67
  5000.5  221.67  5008.5  223.85  5018.5  228.32  5038.5  231.08  5048.5  231.07
  5058.5  232.21  5108.6  230.22  5212.8   239.1  5238.7  241.22  5312.4  243.86
#Mann= 5 ,-1 , 0
  4147.8     .11       0  4848.3     .15       0  4988.5     .09       0
  5018.5     .15       0  5212.8     .11       0
Bank Sta=4988.5,5018.5
XS Rating Curve= 0 ,0
Exp/Cntr=0.3,0.1

Type RM Length L Ch R = 1 ,23658   ,500,500,500
BEGIN DESCRIPTION:
LANDRUM CREEK 43.0
END DESCRIPTION:
XS GIS Cut Line= 3
      3750167.88     10122761.05       3749567.3     10123370.16
      3749167.89     10123711.04
#Sta/Elev= 30
  4144.6  245.09  4331.3  233.31  4370.9  231.18  4434.6  231.32  4469.9  229.66
  4496.2  230.34  4660.9  228.63    4675  228.26    4682  226.23  4703.3  227.65
  4710.3  226.22  4724.5  227.82  4770.1  228.27  4894.2  230.57  4915.4  229.63
    4972  230.56    4979  229.62  4986.2  228.34  4997.1  223.05  5002.9  223.05
  5003.7  221.15  5011.3  221.15  5021.8   226.6 5033.74 229.605  5050.3  230.85
  5156.8  230.31  5241.3  231.79  5367.2  237.57  5440.1     242  5525.1  245.56
#Mann= 7 ,-1 , 0
  4144.6     .11       0  4331.3     .15       0  4496.2     .11       0
  4770.1     .15       0    4979     .09       0 5033.74     .15       0
  5367.2     .11       0
Bank Sta=4979,5033.74
XS Rating Curve= 0 ,0
Exp/Cntr=0.3,0.1

Type RM Length L Ch R = 1 ,23158   ,499,499,499
BEGIN DESCRIPTION:
LANDRUM CREEK 42.0
END DESCRIPTION:
XS GIS Cut Line= 4
      3750267.83     10122611.09      3749503.65     10123096.55
      3749378.46      10123117.7      3749067.82     10122911.05
#Sta/Elev= 30
  3967.7   254.9  4069.3  247.36  4184.5  240.17  4235.1  235.84  4336.1  230.18
  4467.4  228.13  4533.4  228.04  4554.6   225.2    4568  225.21    4597  224.88
  4619.3   229.4  4678.5  230.08  4773.1  229.62  4808.8  228.31  4939.8  229.05
  4980.3  227.75  4987.8  222.96    5000  221.06  5000.8  219.99  5008.8  219.99
  5012.7  225.88 5016.07227.9159  5019.9  230.23  5051.4  230.21    5071  230.84
    5107  229.16  5164.2  232.17  5323.5  233.46  5350.5   234.2  5373.1  237.08
#Mann= 7 ,-1 , 0
  3967.7     .11       0  4235.1     .15       0  4467.4     .11       0
    4568     .15       0  4980.3     .09       0 5016.07     .15       0
  5051.4     .11       0
Bank Sta=4980.3,5016.07
XS Rating Curve= 0 ,0
Exp/Cntr=0.3,0.1

Type RM Length L Ch R = 1 ,22659   ,493,493,493
BEGIN DESCRIPTION:
LANDRUM CREEK 41.0
END DESCRIPTION:
XS GIS Cut Line= 3
      3750067.89     10122211.04      3749466.31     10122704.69
      3749117.84     10122761.07
#Sta/Elev= 30
  4221.8   248.8  4235.5  246.72  4360.9  239.42    4476  228.62  4541.9   225.8
  4591.4  226.95  4712.7  226.27  4797.4   227.9  4896.4  226.31  4953.8  228.45
 4977.19227.6883    4989  225.79  4991.7  221.05  4999.8  221.05  5006.1  223.16
 5014.51227.7728  5018.7  228.87  5079.5   227.6  5109.9   229.1  5129.5   227.9
    5147   228.7  5170.6  228.44  5196.2  225.67  5231.4  225.97  5241.6  226.66
  5251.7  228.94  5302.3  230.45  5319.6  232.97  5324.7   232.7    5353   240.1
#Mann= 6 ,-1 , 0
  4221.8     .11       0  4360.9     .17       0    4476     .15       0
 4977.19     .09       0 5014.51     .15       0    5147     .11       0
Bank Sta=4977.19,5014.51
XS Rating Curve= 0 ,0
Exp/Cntr=0.3,0.1

Type RM Length L Ch R = 1 ,22166   ,437,437,437
BEGIN DESCRIPTION:
LANDRUM CREEK 40.0
END DESCRIPTION:
XS GIS Cut Line= 3
      3750167.83     10122111.08      3749415.38     10122293.76
      3749067.83     10122711.09
#Sta/Elev= 30
  4225.7  256.34    4308  252.94  4410.9  243.79  4431.5  239.75  4441.8  239.04
  4452.1   239.8    4458  242.56  4493.2  239.82  4513.8  236.96  4593.6  231.22
  4708.6  224.11  4740.2  225.85  4904.8  224.77  4976.9  226.65  4987.2  223.88
  4992.1  219.03  5003.5  219.94    5010  224.04  5017.8  226.41  5102.4  226.35
  5110.2  224.44  5152.7  226.82  5180.5   226.6  5188.3  225.14  5223.5  227.86
  5295.1  227.34    5399   229.5  5472.1  232.23  5529.4  246.68  5543.1  245.51
#Mann= 5 ,-1 , 0
  4225.7     .11       0  4593.6     .15       0  4976.9     .09       0
  5017.8     .15       0    5399     .11       0
Bank Sta=4976.9,5017.8
XS Rating Curve= 0 ,0
Exp/Cntr=0.3,0.1

Type RM Length L Ch R = 1 ,21729   ,481,481,481
BEGIN DESCRIPTION:
LANDRUM CREEK 39.0
END DESCRIPTION:
XS GIS Cut Line= 3
      3749867.81     10122111.07      3749232.82     10122008.01
      3748717.88     10122311.06
#Sta/Elev= 30
  4453.6  244.25  4463.7  243.39  4481.8  239.28  4486.9  240.95  4494.1  238.71
  4543.4  230.17  4548.5  230.71  4575.1  228.39  4610.1  228.25  4657.2  225.83
  4794.9  224.46  4970.2  224.65  4984.8  220.34  4986.3  217.15  4994.6  217.15
  5000.6  221.23  5010.8  224.42  5041.1  226.68  5071.5  225.48  5102.7  225.39
  5116.4  226.29  5132.1  225.18  5156.2  225.38  5249.3  225.87  5304.7  227.84
  5446.5  231.07    5474  232.96  5563.6  232.99  5585.1  234.36  5694.4  237.31
#Mann= 6 ,-1 , 0
  4453.6     .11       0  4657.2     .15       0  4970.2     .09       0
  5010.8     .15       0  5156.2     .11       0  5304.7     .17       0
Bank Sta=4970.2,5010.8
XS Rating Curve= 0 ,0
Exp/Cntr=0.3,0.1

Type RM Length L Ch R = 1 ,21248   ,579,579,579
BEGIN DESCRIPTION:
LANDRUM CREEK 38.0
END DESCRIPTION:
XS GIS Cut Line= 3
      3749967.85     10121961.07      3749245.84     10121588.74
      3748628.64     10122104.37
#Sta/Elev= 30
  4351.5  244.94  4359.8  243.94  4365.4  245.74  4404.1  245.01  4409.7  241.54
  4426.2  240.99  4431.9  238.84  4514.9   231.6  4692.2  226.21  4819.6  224.64
  4880.3  223.94  4902.5  225.42  4946.8  224.81  4974.6  226.01  4981.6  225.06
  4991.2  220.47  4992.5  217.24    5001  217.24  5004.1  220.41  5013.3  224.75
  5079.8  225.63  5171.5   223.7  5359.7  224.03  5434.4  223.76  5541.7  225.59
  5590.2  227.92    5640     228    5745  231.18  5760.6  230.45  5968.1  237.42
#Mann= 8 ,-1 , 0
  4351.5     .11       0  4819.6     .15       0  4981.6     .09       0
  5013.3     .15       0  5359.7     .11       0  5541.7     .17       0
  5590.2     .11       0    5745     .17       0
Bank Sta=4981.6,5013.3
XS Rating Curve= 0 ,0
Exp/Cntr=0.3,0.1

Type RM Length L Ch R = 1 ,20669   ,497,497,497
BEGIN DESCRIPTION:
LANDRUM CREEK 37.0
END DESCRIPTION:
XS GIS Cut Line= 3
      3750010.95     10120179.11      3749131.67      10121290.3
      3748517.85     10121911.07
#Sta/Elev= 30
    3583  245.39  3643.6  240.52  3693.3  238.81  3800.7  230.77  3900.1  227.37
  4241.5  223.42  4369.7  224.08    4413  222.86  4448.2   224.2  4776.9  222.91
  4903.4  222.21  4967.5  224.12  4988.3  223.98 4988.84 223.278  4993.9  216.85
  5004.1  216.85  5017.4  218.64  5031.5  223.26    5081  222.64  5137.6  224.32
  5158.8  222.15  5172.9  222.89  5264.9  222.96  5314.4  225.02    5378  225.11
  5554.8  228.85  5667.9  232.86  5795.2  236.01  5852.8  239.69    5873  240.11
#Mann= 5 ,-1 , 0
    3583     .11       0  4776.9     .15       0 4988.84     .09       0
  5031.5     .11       0  5852.8     .17       0
Bank Sta=4988.84,5031.5
XS Rating Curve= 0 ,0
Exp/Cntr=0.3,0.1

Type RM Length L Ch R = 1 ,20172   ,497,497,497
BEGIN DESCRIPTION:
LANDRUM CREEK 36.0
END DESCRIPTION:
XS GIS Cut Line= 3
      3749667.87     10120261.05      3749048.72     10120837.28
      3748467.85     10121311.07
#Sta/Elev= 30
  4154.2  230.21  4267.3  226.21  4451.5  223.11  4585.9  222.97  4642.6  221.61
  4689.3  222.19  4776.9  222.63  4847.8  221.06  4953.8  222.24  4974.8   223.5
 4989.59223.0291  4999.1   217.6  5005.6  217.03  5015.8  217.03  5017.2  219.88
  5025.1  223.02  5130.6  221.43  5159.4  222.78  5188.1  221.99  5223.3  223.01
  5280.7  221.63  5434.2  225.72  5643.3  230.78  5649.8  229.03  5653.4  229.41
  5685.1  229.67  5692.9  230.59  5699.3  232.94  5713.7  234.45  5749.6  232.81
#Mann= 6 ,-1 , 0
  4154.2     .11       0  4689.3     .15       0 4989.59     .09       0
  5025.1     .15       0  5434.2     .17       0  5653.4     .11       0
Bank Sta=4989.59,5025.1
XS Rating Curve= 0 ,0
Exp/Cntr=0.3,0.1

Type RM Length L Ch R = 1 ,19675   ,488,488,488
BEGIN DESCRIPTION:
LANDRUM CREEK 35.0
END DESCRIPTION:
XS GIS Cut Line= 3
      3749517.87     10120111.06      3748742.09     10120525.62
      3748317.87     10120811.06
#Sta/Elev= 30
  4120.4  239.15  4150.5  233.54  4178.1  230.63  4210.7   231.6  4216.3  229.61
  4232.6  232.61  4238.3  230.94  4254.6   232.7  4260.2  230.86  4276.5  231.86
  4282.2  229.56  4298.5  228.87  4304.1  226.53    4348  223.46  4698.5  220.22
    4710  217.12  4732.7  220.02  4836.8  220.57  4880.1  219.52  4978.1  222.63
 4986.69 221.409  4993.5  219.38  4994.5   216.2  5004.7   216.2  5020.9  221.41
  5029.2  222.81  5122.9  220.09  5236.9  219.85  5359.9  223.85  5511.3  231.97
#Mann= 4 ,-1 , 0
  4120.4     .11       0  4836.8     .15       0 4986.69     .09       0
  5020.9     .15       0
Bank Sta=4986.69,5020.9
XS Rating Curve= 0 ,0
Exp/Cntr=0.3,0.1

Type RM Length L Ch R = 1 ,19187   ,494,494,494
BEGIN DESCRIPTION:
LANDRUM CREEK 34.0
END DESCRIPTION:
XS GIS Cut Line= 3
      3749493.62     10120050.62      3748477.98     10120323.29
      3748167.85     10120561.08
#Sta/Elev= 30
  3948.4  239.31  4009.6  232.22  4016.5  228.81  4026.8  226.38  4140.7  226.14
  4159.3  231.53  4171.8  232.48  4192.5  229.37  4199.3  226.63  4213.2  224.32
  4254.6  222.19  4482.4  219.94  4534.2  218.04  4575.6  219.66  4648.1  218.47
  4867.8  219.59  4927.7  219.69  4979.4  221.76  4989.8  219.71  4997.5  214.74
  5000.4  214.21  5010.6  214.21  5012.8  218.65 5016.59219.9133  5034.6  221.16
  5105.2  220.31  5169.6  225.13  5190.4  224.92  5344.6  232.46  5390.8  233.89
#Mann= 5 ,-1 , 0
  3948.4     .11       0  4867.8     .15       0  4989.8     .09       0
 5016.59     .15       0  5344.6     .11       0
Bank Sta=4989.8,5016.59
XS Rating Curve= 0 ,0
Exp/Cntr=0.3,0.1

Type RM Length L Ch R = 1 ,18693   ,468,468,468
BEGIN DESCRIPTION:
LANDRUM CREEK 33.0
END DESCRIPTION:
XS GIS Cut Line= 3
      3749767.83     10120011.07      3748590.18     10119902.91
      3747367.85     10119511.07
#Sta/Elev= 30
  3817.4  249.01  3982.2  244.35    4202  231.71  4339.6  226.03  4399.8  225.12
  4500.2  219.99  4751.5  218.53  4782.9  215.97  4801.5  215.88  4821.6  218.24
    4932  218.41  4966.3  219.99  4987.1  213.49  5020.3  215.06  5025.6  219.31
 5028.63219.9845    5034  221.18  5095.6  220.67  5107.5  221.53  5170.5  219.12
    5244  218.71  5448.5  221.53  5544.9  226.69  5614.4  227.57  5844.6   242.5
  5871.5  245.56  5916.1  246.83  5979.1   251.6  6021.1  252.12  6283.6   263.9
#Mann= 5 ,-1 , 0
  3817.4     .11       0  4782.9     .15       0  4966.3     .09       0
 5028.63     .15       0  5095.6     .11       0
Bank Sta=4966.3,5028.63
XS Rating Curve= 0 ,0
Exp/Cntr=0.3,0.1

Type RM Length L Ch R = 1 ,18225   ,497,497,497
BEGIN DESCRIPTION:
LANDRUM CREEK 32.0
END DESCRIPTION:
XS GIS Cut Line= 3
      3749667.83     10119911.07      3748545.51     10119600.51
      3747667.85     10119511.07
#Sta/Elev= 30
  3835.5  250.25  4079.3  237.95  4105.3  234.79  4323.1  222.73  4406.2  220.16
  4582.6  217.19  4665.5  217.99  4680.1  217.12  4686.3  214.89  4696.7  215.36
    4707  217.78  4714.5  218.13  4727.8  217.46  4873.1  218.69  4914.6  217.88
  4966.4  219.09  4975.4  216.29  4980.6  218.71    4991  213.15  5001.3  213.15
  5007.7  216.59  5017.7  216.97 5024.34218.7779  5027.8  219.72  5044.4     219
  5188.6  217.67  5409.8  221.39  5610.8  233.54  5791.7  248.17  5882.2  252.75
#Mann= 5 ,-1 , 0
  3835.5     .11       0  4582.6     .15       0  4980.6     .09       0
 5024.34     .15       0  5044.4     .11       0
Bank Sta=4980.6,5024.34
XS Rating Curve= 0 ,0
Exp/Cntr=0.3,0.1

Type RM Length L Ch R = 1 ,17728   ,489,489,489
BEGIN DESCRIPTION:
LANDRUM CREEK 31.0
END DESCRIPTION:
XS GIS Cut Line= 3
      3749635.94      10119741.6      3748235.09     10119259.16
      3747917.89     10119261.07
#Sta/Elev= 30
  3518.4  249.35    3565  246.09  3627.5  238.79  3658.7  238.86  3706.8   234.3
  3778.3  233.33  3823.1  228.99  3908.5  226.41  3991.5   221.3  4078.5  219.55
  4209.1  216.81  4235.6  217.43  4277.9  214.68  4298.4  217.86  4333.8  217.17
  4381.2  216.94  4468.3   217.4  4510.6  214.51    4518  215.59    4621  217.84
    4724  217.14  4758.5  217.49    4930  218.14    4980  218.42  4990.7   211.9
    5001   211.9 5015.62218.3416  5037.2  221.79  5097.2   226.4  5317.2  240.28
#Mann= 12 ,-1 , 0
  3518.4     .11       0  4078.5     .17       0  4209.1     .15       0
  4333.8     .11       0  4381.2     .15       0    4518     .17       0
    4621     .15       0    4724     .17       0  4758.5     .15       0
    4930     .11       0    4980     .06       0 5015.62     .11       0
Bank Sta=4980,5015.62
XS Rating Curve= 0 ,0
Exp/Cntr=0.3,0.1

Type RM Length L Ch R = 1 ,17239   ,485,485,485
BEGIN DESCRIPTION:
LANDRUM CREEK 30.0
END DESCRIPTION:
XS GIS Cut Line= 3
      3749417.84     10119611.06      3748511.14     10118886.89
      3747831.59     10118540.82
#Sta/Elev= 30
  3839.6  235.09  3906.7  230.35  3989.3  227.23  4016.6  224.85  4072.2  222.31
  4123.7  221.06  4351.5   216.8  4493.6  216.57  4565.7  214.96  4629.1  215.81
  4734.3  215.79  4985.2  216.18  4986.4  213.33  4996.7  213.33  5004.5216.1997
  5059.8  218.25  5066.7  215.38  5072.3  215.01  5092.6  217.28  5105.6  217.36
  5321.5  221.16    5327  221.27  5461.4  224.45    5467  225.96  5511.5  228.24
  5561.4   227.4  5572.6  226.39  5648.6  228.75  5757.2  233.15  5762.6  233.16
#Mann= 16 ,-1 , 0
  3839.6     .11       0  3906.7     .17       0  4016.6     .11       0
  4072.2     .17       0  4123.7     .11       0  4629.1     .15       0
  4734.3     .17       0  4985.2     .09       0  5004.5     .17       0
  5092.6     .15       0  5105.6     .17       0  5321.5     .11       0
    5327     .17       0  5561.4     .11       0  5648.6     .17       0
  5757.2     .11       0
Bank Sta=4985.2,5004.5
XS Rating Curve= 0 ,0
Exp/Cntr=0.3,0.1

Type RM Length L Ch R = 1 ,16754   ,498,498,498
BEGIN DESCRIPTION:
LANDRUM CREEK 29.0
END DESCRIPTION:
XS GIS Cut Line= 3
      3749667.85     10118911.07      3748768.71     10118539.74
      3748093.59     10118325.82
#Sta/Elev= 30
  4027.2  245.67  4095.1  243.18  4355.9  225.45  4373.4  221.25  4379.8  217.94
  4403.8  213.91  4416.7  213.25    4457  213.37  4503.2  224.45  4557.3  215.99
  4693.3  213.85  4723.2  213.27  4736.1  210.89  4746.4  210.89  4747.2  213.14
  4771.1  215.08  4954.7  215.42  4984.1  216.66  4990.1  214.62  5003.1  213.57
  5009.1  215.73  5014.4  214.95  5021.9  216.83  5116.5   214.8  5245.6  216.21
  5263.2  215.01  5315.6  215.37  5376.5  216.89  5476.9  219.62  5708.2   231.8
#Mann= 5 ,-1 , 0
  4027.2     .11       0  4693.3     .15       0  4723.2     .09       0
  4747.2     .15       0  5376.5     .17       0
#Block Obstruct= 2 , 0
         4501.71  224.41
Bank Sta=4723.2,4747.2
XS Rating Curve= 0 ,0
Exp/Cntr=0.3,0.1

Type RM Length L Ch R = 1 ,16256   ,499,499,499
BEGIN DESCRIPTION:
LANDRUM CREEK 28.0
END DESCRIPTION:
XS GIS Cut Line= 3
      3749639.39     10118620.06      3748557.87     10118151.89
      3748199.41     10118095.92
#Sta/Elev= 30
  3821.5  236.59  3866.8  232.75  3964.8  228.01  4073.8  219.49  4318.9  212.98
  4390.3  214.16 4407.83  213.16  4426.7   210.1    4437   210.1  4444.3  213.13
    4636  215.05  4651.3  213.39  4688.4  215.34  4793.3  214.92  4811.3  213.37
  4916.1  214.94  4963.1  214.69  4986.6  211.66  5002.5  211.73  5030.4  212.95
  5041.6  215.04  5091.1  215.42  5099.3  217.11  5104.4  216.36  5151.8  219.55
  5182.2     223  5202.4   221.4    5253  225.68  5333.3  228.52  5362.8  230.57
#Mann= 5 ,-1 , 0
  3821.5     .11       0  4318.9     .15       0 4407.83     .09       0
  4444.3     .15       0  5333.3     .17       0
Bank Sta=4407.83,4444.3
XS Rating Curve= 0 ,0
Exp/Cntr=0.3,0.1

Type RM Length L Ch R = 1 ,15757   ,487,487,487
BEGIN DESCRIPTION:
LANDRUM CREEK 27.0
END DESCRIPTION:
XS GIS Cut Line= 3
      3750067.89     10117561.06      3748848.48     10117853.13
      3748267.82     10117611.06
#Sta/Elev= 30
  3746.1  255.46  3769.7  254.53  3848.6  247.38  3853.8  247.87  3895.8  242.62
  3937.8  238.88    3943  239.95  3974.7  236.62  4000.8  233.49  4063.9  228.02
  4069.1  229.14  4077.1   228.5  4153.1  221.57    4178  221.41  4195.2  218.48
  4229.4  215.63  4368.4  211.96  4620.2  211.06  4980.1  214.07  4990.4  213.25
  4992.6  210.24  5002.9  210.24  5011.5  212.98  5070.7  213.83  5147.6  212.68
  5210.1  214.86  5293.2  217.85    5369   222.7  5596.4  233.83  5629.1  234.65
#Mann= 8 ,-1 , 0
  3746.1     .17       0  3974.7     .11       0  4000.8     .17       0
  4077.1     .15       0  4990.4     .09       0  5011.5     .15       0
  5210.1     .17       0  5596.4     .15       0
Bank Sta=4990.4,5011.5
XS Rating Curve= 0 ,0
Exp/Cntr=0.3,0.1

Type RM Length L Ch R = 1 ,15270   ,558,558,558
BEGIN DESCRIPTION:
LANDRUM CREEK 26.0
END DESCRIPTION:
XS GIS Cut Line= 3
      3750167.81     10117511.07      3748972.45     10117492.83
      3748367.85     10117411.07
#Sta/Elev= 30
  3804.5   263.4    3858  259.69  3924.5  254.75  3984.5  248.45  4045.9  243.51
  4249.1  224.14  4324.5  212.84  4404.5  210.74  4484.5  211.16  4584.6  210.43
  4609.4  207.07  4619.7  207.07  4634.6  210.74  4824.6  210.81  4944.6  212.66
  4964.6  212.31  4974.6  211.51  4984.6  209.57  5024.8  213.01  5063.9   212.8
  5110.5  212.63  5211.4  214.76  5307.4  219.34  5337.6  220.59  5418.4  226.83
  5478.9  228.71  5496.1  230.46  5501.2  229.79  5519.3  230.14  5610.1  233.88
#Mann= 10 ,-1 , 0
  3804.5     .11       0    3858     .17       0  4045.9     .11       0
  4249.1     .15       0  4584.6     .09       0  4634.6     .15       0
  5063.9     .11       0  5110.5     .17       0  5211.4     .15       0
  5307.4     .17       0
Bank Sta=4584.6,4634.6
XS Rating Curve= 0 ,0
Exp/Cntr=0.3,0.1

Type RM Length L Ch R = 1 ,14712   ,727,727,727
BEGIN DESCRIPTION:
LANDRUM CREEK 25.0
END DESCRIPTION:
XS GIS Cut Line= 3
      3750267.83     10117461.06      3749184.56     10116984.66
      3748649.85      10116380.5
#Sta/Elev= 30
  3819.6  267.73  3857.3  267.15  3994.4  258.35  4267.5  229.92  4380.3  221.19
  4450.4  213.22  4502.5  210.64  4549.2  210.15  4562.4  208.54  4572.5  209.54
    4578  208.53  4584.3  209.82  4676.8   209.6  4688.4  206.75  4698.7  206.75
  4700.2  208.97  4715.4  209.62  4897.9  210.91  4940.9  208.38    4950  209.87
  4973.4  209.75  4978.8  211.88  5001.2  208.22  5008.5  209.61  5024.2  212.09
  5201.6  210.17  5336.2  213.21    5414  213.44  5740.2  229.34  5809.8  235.54
#Mann= 5 ,-1 , 0
  3819.6     .11       0  4676.8     .09       0  4715.4     .11       0
  4940.9     .15       0  5008.5     .11       0
Bank Sta=4676.8,4715.4
XS Rating Curve= 0 ,0
Exp/Cntr=0.3,0.1
