HEC-RAS study LITTLE CANEY CREEK.prj: LITTLE CANEY CREEK Base Level Engineering

--- LITTLE CANEY CREEK.g01 (geometry) --- (continued)

Type RM Length L Ch R = 1 ,64025   ,631,631,631
BEGIN DESCRIPTION:
LITTLE CANEY CREEK 81.0
END DESCRIPTION:
XS GIS Cut Line= 3
      3706767.83     10154461.03      3705976.49     10152915.21
      3706617.85     10151311.07
#Sta/Elev= 30
  3263.4  299.08  3279.7  298.73  3445.8  290.62  3643.5  276.49  3720.3   268.2
  3782.4  263.41  4006.9  262.05    4204  262.28  4787.1  262.73  4853.7  259.03
  4892.3  263.09  4914.7  263.19  4964.1  260.58  4981.3     263 4986.22260.3905
  4992.7  256.17  5006.3  256.17  5013.5  260.46  5018.9   258.7    5026  261.13
  5058.3  261.97  5236.2  263.76  5336.6  264.07  5527.9   273.2  5748.7  273.28
  6012.6  278.63  6221.4  278.74  6385.5  282.11  6561.9  284.88  6727.6  289.48
#Mann= 11 ,-1 , 0
  3263.4     .11       0  3279.7     .17       0  3445.8     .11       0
  3720.3     .15       0  4006.9     .11       0    4204     .15       0
 4986.22     .09       0  5013.5     .15       0  5236.2     .11       0
  6385.5     .17       0  6561.9     .11       0
Bank Sta=4986.22,5013.5
XS Rating Curve= 0 ,0
Exp/Cntr=0.3,0.1

Type RM Length L Ch R = 1 ,63394   ,467,467,467
BEGIN DESCRIPTION:
LITTLE CANEY CREEK 80.0
END DESCRIPTION:
XS GIS Cut Line= 3
      3706867.86     10154111.09      3706535.06     10153091.93
      3707097.55     10151461.76
#Sta/Elev= 30
    3849  293.84  3902.1  294.02  3985.8  290.69  4185.2  270.18  4259.3  264.43
  4385.7  260.38  4595.9  262.91  4704.6  262.47  4722.1  259.93  4743.2  262.13
  4806.3  260.07  4879.9  261.75  4985.5   260.7  4989.3  255.92  5002.9  255.92
  5017.2  261.48  5144.2  261.66  5207.6  259.25  5302.9  262.49  5334.6  260.61
  5422.7   267.2  5472.1  271.88  5510.6  272.36  5659.2  275.55    5898  281.51
  5931.2  279.41  6159.7  278.33  6261.8  280.67  6443.6  280.21  6645.6  283.43
#Mann= 8 ,-1 , 0
    3849     .17       0  4185.2     .15       0  4985.5     .09       0
  5017.2     .15       0  5422.7     .17       0  5510.6     .11       0
  5659.2     .17       0  5931.2     .11       0
Bank Sta=4985.5,5017.2
XS Rating Curve= 0 ,0
Exp/Cntr=0.3,0.1

Type RM Length L Ch R = 1 ,62927   ,598,598,598
BEGIN DESCRIPTION:
LITTLE CANEY CREEK 79.0
END DESCRIPTION:
XS GIS Cut Line= 3
      3707087.14     10154055.43      3706993.53     10153111.06
       3707118.4     10151560.68
#Sta/Elev= 30
    4051  291.43  4235.9   279.5  4326.7  270.48  4427.3  265.97  4618.1  259.87
  4768.9  261.35    4789  260.37  4819.1  262.03  4989.9  260.28  5002.5  258.99
  5002.7  255.03  5003.2  254.53  5016.8  254.53  5020.1  257.85  5030.1  259.98
    5321  261.66  5365.7  260.75  5371.2  259.16  5391.3  260.73  5441.4  259.78
  5451.4  260.32  5471.5  265.92  5514.7  267.89  5652.1  270.17  5752.4   274.5
  5953.1  279.95  6067.3  279.89    6244  279.04  6394.5  282.25  6555.4  281.71
#Mann= 7 ,-1 , 0
    4051     .17       0  4235.9     .11       0  4427.3     .15       0
  4989.9     .09       0  5030.1     .15       0  5514.7     .17       0
  6067.3     .11       0
Bank Sta=4989.9,5030.1
XS Rating Curve= 0 ,0
Exp/Cntr=0.3,0.1

Type RM Length L Ch R = 1 ,62329   ,656,656,656
BEGIN DESCRIPTION:
LITTLE CANEY CREEK 78.0
END DESCRIPTION:
XS GIS Cut Line= 3
      3707267.86     10154161.05      3707514.19     10153043.28
      3707417.85     10151611.11
#Sta/Elev= 30
  3855.4  292.86  3874.7  293.88  3948.4  290.91  4039.7  288.05  4073.5   285.5
  4157.4  281.39  4288.3  277.01  4336.7  275.33    4521  274.45  4703.9  263.87
  4787.2  259.94  4971.5  259.97  4981.8  254.27  4988.7  252.28  5002.3  252.28
  5002.8  252.78  5003.6  258.23  5018.6  260.31  5023.6  259.08  5032.3  260.23
  5202.7  260.59    5373  259.07  5423.2  262.78  5518.2  263.47  5603.6  261.18
  5663.7  262.01  6020.5  273.98  6050.5  274.95  6281.5   280.2  6435.4  283.55
#Mann= 12 ,-1 , 0
  3855.4     .11       0  3948.4     .17       0  4073.5     .11       0
  4157.4     .17       0  4288.3     .11       0  4703.9     .15       0
  4971.5     .09       0  5018.6     .15       0  5518.2     .17       0
  6020.5     .11       0  6050.5     .17       0  6281.5     .11       0
Bank Sta=4971.5,5018.6
XS Rating Curve= 0 ,0
Exp/Cntr=0.3,0.1

Type RM Length L Ch R = 1 ,61673   ,722,722,722
BEGIN DESCRIPTION:
LITTLE CANEY CREEK 77.0
END DESCRIPTION:
XS GIS Cut Line= 3
      3707867.85     10154061.07      3708035.06     10152977.35
      3708321.51     10151701.35
#Sta/Elev= 30
  3901.4  286.96  3998.6  284.83  4075.3  281.06  4086.6   280.7  4275.8  274.34
  4455.8  272.43    4611  269.02  4723.6  266.33  4822.2  260.82  4933.5  259.92
  4973.9  261.27  4986.3  259.69  4997.5  253.08  5011.2  253.08  5014.6  256.27
  5031.8  259.03  5045.4  257.56  5178.6  260.82    5406  262.25  5455.3  262.96
  5475.8  261.44  5496.3   263.5  5598.8  264.35  5685.8   270.4  5752.5  274.74
    5898  277.99  5967.8  276.51  5998.5  277.78  6127.9  277.25  6305.7  281.16
#Mann= 9 ,-1 , 0
  3901.4     .11       0  4075.3     .17       0  4086.6     .11       0
    4611     .15       0  4986.3     .09       0  5031.8     .15       0
    5406     .11       0  5685.8     .17       0    5898     .11       0
Bank Sta=4986.3,5031.8
XS Rating Curve= 0 ,0
Exp/Cntr=0.3,0.1

Type RM Length L Ch R = 1 ,60951   ,1500,1500,1500
BEGIN DESCRIPTION:
LITTLE CANEY CREEK 76.0
END DESCRIPTION:
XS GIS Cut Line= 3
      3708305.89     10154310.72       3708618.4     10152909.64
      3709092.16     10151415.46
#Sta/Elev= 30
  3813.2  289.52  3925.5  288.65  4166.5  276.61  4355.9  270.28  4478.8  271.75
  4718.5  264.41  4980.9  258.59    4988  251.44  5001.7  251.44  5011.6  258.86
  5062.8  261.05  5081.8  259.29  5103.8   261.4    5196  258.63  5216.5  261.67
  5397.6  258.19  5834.7  258.42  5989.1  261.16  6085.9   267.4  6117.9   265.7
  6128.7  262.25  6180.9  266.24  6386.9  268.66  6451.5  267.25  6483.7  270.28
    6611  273.21  6691.9  277.77  6728.5  281.91  6803.8  284.45  6816.2  285.09
#Mann= 7 ,-1 , 0
  3813.2     .11       0  4718.5     .15       0  4980.9     .09       0
  5011.6     .15       0  6691.9     .17       0  6728.5     .11       0
  6803.8     .17       0
Bank Sta=4980.9,5011.6
XS Rating Curve= 0 ,0
Exp/Cntr=0.3,0.1

Type RM Length L Ch R = 1 ,59451   ,679,679,679
BEGIN DESCRIPTION:
LITTLE CANEY CREEK 75.0
END DESCRIPTION:
XS GIS Cut Line= 3
      3708831.95     10154404.41      3709706.94      10152883.6
      3709769.37     10151364.44
#Sta/Elev= 30
  3156.9  282.36  3494.6  272.82    3624  272.54  3661.3  269.51  3682.9  271.99
  4015.2  269.07  4266.1  264.01  4520.2   262.6  4657.8  259.09  4782.3  255.69
  4798.1  258.16    4974  259.21  4984.1  256.34  4987.2  250.44    5001  250.44
  5014.1  257.56  5034.1  259.13  5254.3  258.37  5284.3  255.21  5314.3  258.17
  5599.5  262.86  5787.9   270.8  5961.3   272.7  6044.9  273.99    6075  270.21
    6105  273.24    6135  271.46  6185.1  276.28  6333.1  278.86  6431.9  281.69
#Mann= 10 ,-1 , 0
  3156.9     .11       0  4015.2     .17       0  4266.1     .11       0
  4520.2     .17       0  4657.8     .15       0    4974     .09       0
  5034.1     .15       0  5599.5     .17       0  5961.3     .11       0
  6333.1     .17       0
Bank Sta=4974,5034.1
XS Rating Curve= 0 ,0
Exp/Cntr=0.3,0.1

Type RM Length L Ch R = 1 ,58772   ,406,406,406
BEGIN DESCRIPTION:
LITTLE CANEY CREEK 74.0
END DESCRIPTION:
XS GIS Cut Line= 3
      3708941.34     10154560.65      3710087.15     10153201.31
      3710352.79     10152378.34
#Sta/Elev= 30
  3331.7  283.98  3598.5   276.2    3648  276.37  3711.7   273.1    3748  274.36
  3904.1  273.74  4037.4  271.05  4187.6  267.62  4300.8  269.95  4407.4  270.45
  4528.3  264.29  4606.3  262.45  4854.7  262.28  4880.5  261.31  4961.3  257.78
  4967.9  255.28  4975.6  249.74    4983  248.39  4996.8  248.39  5010.8  258.37
  5031.6  260.13  5067.9  258.15  5172.8  259.24  5246.4  257.25  5761.3  257.53
  5778.1  258.79  5824.3  268.04  5907.7  275.57  5971.4  277.39  5974.3  277.39
#Mann= 7 ,-1 , 0
  3331.7     .11       0  4037.4     .17       0  4880.5     .15       0
  4961.3     .09       0  5010.8     .15       0  5907.7     .17       0
  5971.4     .15       0
Bank Sta=4961.3,5010.8
XS Rating Curve= 0 ,0
Exp/Cntr=0.3,0.1

Type RM Length L Ch R = 1 ,58366   ,622,622,622
BEGIN DESCRIPTION:
LITTLE CANEY CREEK 73.0
END DESCRIPTION:
XS GIS Cut Line= 3
       3709285.1     10154524.19      3710357.98     10153451.31
      3710367.85     10152461.04
#Sta/Elev= 30
  3405.3  278.36  3850.9  268.68  3975.1  269.57  4031.7  267.57  4102.4  269.89
  4136.7   269.1  4328.7  269.29    4463  267.44  4547.2  260.73    4661  255.35
  4682.2  257.56  4731.7  258.83  4851.9  257.46  4963.7  257.89  4982.8  256.29
  5005.9  250.42  5019.7  250.42  5042.8   255.7  5052.8  256.56  5122.8  258.52
  5182.8  256.99  5482.8  256.47  5622.9  257.74  5652.9  256.44  5732.9  256.58
  5772.9  260.16  5792.9  264.91  5832.9  269.64  5905.8  274.41  5912.9  274.69
#Mann= 8 ,-1 , 0
  3405.3     .11       0  3850.9     .15       0  4136.7     .17       0
  4547.2     .11       0  4963.7     .15       0  4982.8     .09       0
  5052.8     .15       0  5905.8     .17       0
Bank Sta=4982.8,5052.8
XS Rating Curve= 0 ,0
Exp/Cntr=0.3,0.1

Type RM Length L Ch R = 1 ,57744   ,440,440,440
BEGIN DESCRIPTION:
LITTLE CANEY CREEK 72.0
END DESCRIPTION:
XS GIS Cut Line= 3
      3709267.86     10154711.06      3710852.93     10153297.83
      3710917.85     10151861.09
#Sta/Elev= 30
  2876.4  286.62  2940.3   284.4  3003.9  280.18    3457  268.02  3556.5  267.19
  3875.1  269.24    4109  257.12  4215.4  255.78    4243  257.46  4533.9  256.21
  4646.8  257.64  4803.1  256.37  4966.1  257.57  4993.1  249.82  5006.9  249.82
  5016.8  257.35  5023.1  257.11  5096.9  256.04  5121.4  254.32  5156.9  251.54
  5186.9  255.91  5367.1  264.52    5416  264.67  5547.3  267.19  5707.5  267.38
  5806.2  270.32  5907.2   271.8  6103.6  277.73  6300.1  288.02  6438.2  294.12
#Mann= 10 ,-1 , 0
  2876.4     .11       0  4966.1     .06       0  5016.8     .11       0
  5023.1     .15       0  5121.4     .11       0    5416     .17       0
  5806.2     .15       0  5907.2     .17       0  6103.6     .15       0
  6300.1     .17       0
Bank Sta=4966.1,5016.8
XS Rating Curve= 0 ,0
Exp/Cntr=0.3,0.1

Type RM Length L Ch R = 1 ,57304   ,654,654,654
BEGIN DESCRIPTION:
LITTLE CANEY CREEK 71.0
END DESCRIPTION:
XS GIS Cut Line= 3
      3709446.54     10154685.67       3711118.4     10153670.06
      3711092.37     10152035.32
#Sta/Elev= 30
  2980.6  279.93  3216.5  272.01  3421.9  267.21  3596.3  268.43  3939.3  255.96
    4788  255.39  4975.7  257.49  4985.8  254.54  4988.9  249.72  5002.7  249.72
  5005.8  253.61  5015.8  256.55  5045.8  257.51  5125.4   256.8  5315.8  257.09
  5355.8  255.33  5385.8  251.27  5405.8  256.33  5525.8  262.21  5665.8  267.33
  5715.6     266  5765.8  266.93  5785.9   265.5  5826.6  265.78    5912  264.11
  5955.9  266.22  6026.4     267  6335.9  273.99  6355.9  273.17  6571.7  279.39
#Mann= 8 ,-1 , 0
  2980.6     .11       0    4788     .15       0  4975.7     .09       0
  5045.8     .15       0  5125.4     .11       0  5715.6     .15       0
  5826.6     .11       0  6026.4     .15       0
Bank Sta=4975.7,5045.8
XS Rating Curve= 0 ,0
Exp/Cntr=0.3,0.1

Type RM Length L Ch R = 1 ,56650   ,593,593,593
BEGIN DESCRIPTION:
LITTLE CANEY CREEK 70.0
END DESCRIPTION:
XS GIS Cut Line= 3
      3709317.82     10154961.09      3711321.57     10153967.21
      3711717.86     10151561.02
#Sta/Elev= 30
  2763.3  289.15  2934.2  285.55  3075.9  277.36  3455.4  266.15  3622.9  266.31
  3657.1  270.38  3673.9  266.94  3875.7  256.28  4204.5  256.78  4296.3  256.12
  4605.5  254.45  4917.9  253.52  4979.6  255.82  4988.2  249.79  5002.1  249.79
  5026.5   256.5  5621.3  255.47  5654.8  252.55  5682.5  255.85  5809.9  255.85
  5877.1  258.51  5930.3  259.48  6075.1   259.2  6374.4  262.92  6732.5  271.21
  6916.1  272.07  6995.2  275.49  7185.2  286.39  7221.9   291.2  7438.6  302.08
#Mann= 10 ,-1 , 0
  2763.3     .11       0  4204.5     .17       0  4296.3     .11       0
  4605.5     .15       0  4979.6     .09       0  5026.5     .15       0
  5877.1     .17       0  5930.3     .15       0  6075.1     .17       0
  6995.2     .11       0
Bank Sta=4979.6,5026.5
XS Rating Curve= 0 ,0
Exp/Cntr=0.3,0.1

Type RM Length L Ch R = 1 ,56057   ,613,613,613
BEGIN DESCRIPTION:
LITTLE CANEY CREEK 69.0
END DESCRIPTION:
XS GIS Cut Line= 3
      3711217.85     10155361.08       3711759.9     10153978.97
      3712867.85     10152361.08
#Sta/Elev= 30
  3515.4  276.71  3934.3  260.93  4018.5  260.61  4023.9  262.75  4033.7  260.94
  4078.1  261.39    4127  258.01  4216.4  262.79  4317.9  259.37  4355.9  258.21
    4564  255.23  4880.1  255.06  4975.8  255.63  4989.2  247.39  5003.2  247.39
  5004.4  250.87  5010.4  256.27  5126.4  254.76  5164.4  253.54  5688.3  254.96
  5709.8  253.04  6159.3  257.42  6245.1  258.98  6258.6  260.03  6403.1  268.36
  6615.3   272.3  6718.5  274.37  6800.5  276.79  6826.5  277.65  6960.9  280.93
#Mann= 18 ,-1 , 0
  3515.4     .11       0  4033.7     .17       0  4317.9     .11       0
  4355.9     .15       0    4564     .11       0  4880.1     .15       0
  4975.8     .09       0  5010.4     .15       0  5126.4     .11       0
  5164.4     .15       0  6159.3     .11       0  6245.1     .17       0
  6258.6     .11       0  6403.1     .17       0  6615.3     .11       0
  6718.5     .17       0  6800.5     .11       0  6826.5     .17       0
Bank Sta=4975.8,5010.4
XS Rating Curve= 0 ,0
Exp/Cntr=0.3,0.1

Type RM Length L Ch R = 1 ,55444   ,485,485,485
BEGIN DESCRIPTION:
LITTLE CANEY CREEK 68.0
END DESCRIPTION:
XS GIS Cut Line= 3
      3712054.16     10155540.74      3712106.24     10153962.59
      3712767.83     10152711.11
#Sta/Elev= 30
  3708.7  275.62  3908.5  268.41  4083.2  265.08  4208.6   262.7  4453.2  264.49
  4588.9  263.74  4711.3  265.92  4715.1  265.91  4758.9  265.34  4865.9     260
    4939  255.17  4979.1  255.46  4989.1  253.36  4992.1  247.65  5006.1  247.65
  5009.1  250.91  5019.1  254.96  5143.4  254.83  5338.4  252.99  5451.6  253.03
  5514.7  253.51  5985.8  254.52    6002  252.78  6013.5  254.43  6214.3  255.33
  6323.3  258.23  6392.7  260.28  6502.7  267.08  6541.1  267.18  6703.3  274.24
#Mann= 14 ,-1 , 0
  3708.7     .11       0  4083.2     .15       0  4453.2     .17       0
  4711.3     .11       0  4715.1     .17       0  4865.9     .15       0
  4979.1     .09       0  5019.1     .15       0  5143.4     .11       0
  5338.4     .15       0  5451.6     .11       0  5514.7     .15       0
  6214.3     .11       0  6323.3     .17       0
Bank Sta=4979.1,5019.1
XS Rating Curve= 0 ,0
Exp/Cntr=0.3,0.1

Type RM Length L Ch R = 1 ,54959   ,387,387,387
BEGIN DESCRIPTION:
LITTLE CANEY CREEK 67.0
END DESCRIPTION:
XS GIS Cut Line= 3
      3712217.85     10155561.07      3712446.79     10153987.84
      3712817.85     10152861.06
#Sta/Elev= 30
  3410.2   276.6  3580.4  268.43  3777.9  264.09  3843.8  263.71  4034.9  261.89
  4127.7  261.35  4299.5  266.34  4380.8  266.27  4546.4  258.23  4582.4  254.98
  4666.8  253.74  4765.6  253.48  4767.7  253.47  4963.2  254.35  4986.6  255.12
  4995.8  252.62  5000.1   247.5  5014.1   247.5  5015.9  250.97  5021.1  248.03
  5038.7  254.47  5084.7   251.8    5165  251.27  5693.7  252.86  5779.4  254.97
  5881.6  260.23  5983.8  267.11  5985.3  267.27  6106.8   273.2  6186.3  274.55
#Mann= 16 ,-1 , 0
  3410.2     .11       0  3777.9     .15       0  3843.8     .11       0
  4034.9     .17       0  4380.8     .11       0  4546.4     .15       0
  4666.8     .17       0  4765.6     .15       0  4767.7     .11       0
  4963.2     .15       0  4986.6     .09       0  5038.7     .15       0
  5779.4     .11       0  5881.6     .17       0  5983.8     .11       0
  5985.3     .17       0
Bank Sta=4986.6,5038.7
XS Rating Curve= 0 ,0
Exp/Cntr=0.3,0.1

Type RM Length L Ch R = 1 ,54572   ,608,608,608
BEGIN DESCRIPTION:
LITTLE CANEY CREEK 66.0
END DESCRIPTION:
XS GIS Cut Line= 4
      3712619.58     10155222.31      3712482.01     10154632.22
      3712741.66     10154103.22      3712877.08     10153056.34
#Sta/Elev= 30
       0  267.74    62.9  267.02    83.4  265.22     104   266.1   251.4   263.7
   432.5  259.18   545.5  265.27   605.9  265.38   685.2  261.42   722.7  258.81
     752  256.58   829.6  253.97  1133.1  253.36  1155.6  251.72    1178  254.26
  1186.5  249.71  1193.6   248.7  1198.8   248.7  1203.4  252.58  1208.5   251.4
  1217.5   253.8  1499.9  252.52  1669.2  252.86  1711.6     252  1731.8  250.11
    1762  251.75  1893.1  251.91    2004  256.67  2074.6  262.78  2250.8  272.18
#Mann= 8 ,-1 , 0
       0     .11       0   251.4     .15       0   605.9     .11       0
   685.2     .15       0   722.7     .11       0    1178     .06       0
  1217.5     .15       0  1499.9     .11       0
Bank Sta=1178,1217.5
XS Rating Curve= 0 ,0
Exp/Cntr=0.3,0.1

Type RM Length L Ch R = 1 ,53964   ,565,565,565
BEGIN DESCRIPTION:
LITTLE CANEY CREEK 65.0
END DESCRIPTION:
XS GIS Cut Line= 3
      3712845.74     10155514.27      3713114.31     10153967.49
      3712917.85     10153061.07
#Sta/Elev= 30
       0   269.7   165.6  266.92   278.9   266.6   348.3  263.82   480.3  261.35
     866  257.72   957.3  258.45  1153.7  260.58  1327.7   255.5  1382.3  252.06
  1535.8  253.03  1556.1  251.96  1561.3   246.7  1569.9  247.04  1574.1   249.7
  1579.2  249.41  1586.7  252.74  1607.2  253.54  1637.9  251.76  1908.2  251.48
  1924.4  248.93  1957.3   252.3  2143.8  251.25  2159.7  252.51  2180.2   251.2
  2187.9  251.53  2200.7  254.76  2272.3  258.44  2384.8  267.13  2497.4     271
#Mann= 5 ,-1 , 0
       0     .11       0   957.3     .15       0  1556.1     .09       0
  1586.7     .15       0  1908.2     .11       0
Bank Sta=1556.1,1586.7
XS Rating Curve= 0 ,0
Exp/Cntr=0.3,0.1

Type RM Length L Ch R = 1 ,53399   ,533,533,533
BEGIN DESCRIPTION:
LITTLE CANEY CREEK 64.0
END DESCRIPTION:
XS GIS Cut Line= 3
      3713467.85     10155611.06       3713517.7      10153845.4
      3713830.21     10152876.62
#Sta/Elev= 30
  3425.2  273.45  3505.2  272.66  3905.4  263.16  4085.4  260.71  4155.5  260.16
  4255.5  263.77  4315.8  259.15  4775.7  260.44  4935.8  256.15  4965.8  254.95
  4975.8  253.14  4985.8  249.55  4988.8  245.33  5002.8  245.33  5005.8  250.18
  5015.2  253.44  5055.8   251.7  5217.1  251.26  5236.9   252.2  5562.6  250.28
  5574.4   248.6  5713.9  253.53    5753  255.63  5837.1   264.6    5904  269.31
  5957.7   271.6  5973.7  270.38  6027.1  273.96  6117.5  276.09  6209.5  279.66
#Mann= 7 ,-1 , 0
  3425.2     .11       0  4935.8     .15       0  4975.8     .09       0
  5015.2     .15       0  5713.9     .11       0    5904     .17       0
  6117.5     .11       0
Bank Sta=4975.8,5015.2
XS Rating Curve= 0 ,0
Exp/Cntr=0.3,0.1

Type RM Length L Ch R = 1 ,52866   ,330,330,330
BEGIN DESCRIPTION:
LITTLE CANEY CREEK 63.0
END DESCRIPTION:
XS GIS Cut Line= 3
      3713637.38      10155377.1      3713911.95     10153827.03
      3713908.33     10153040.74
#Sta/Elev= 30
  3425.8  269.32  3899.1  259.34  4033.3  257.92  4318.8  257.16  4366.2  258.59
  4491.2  256.57  4731.8  256.62  4843.6  251.68  4863.9  249.02    4895  249.27
  4918.7  251.39  4985.7  251.35  4995.4  246.33    5006  245.41    5016  250.72
    5026  251.22    5076  251.87    5176  249.64    5196  246.68    5256   246.3
    5269  244.64    5283  244.64    5296  246.55    5306  249.88    5336  256.16
  5356.3  256.73    5416  260.82    5556  264.33  5683.8  270.29  5786.3  274.79
#Mann= 6 ,-1 , 0
  3425.8     .11       0  4918.7     .15       0    5176     .09       0
    5306     .15       0  5356.3     .11       0  5683.8     .17       0
Bank Sta=5176,5306
XS Rating Curve= 0 ,0
Exp/Cntr=0.3,0.1

Type RM Length L Ch R = 1 ,52536   ,666,666,666
BEGIN DESCRIPTION:
LITTLE CANEY CREEK 62.0
END DESCRIPTION:
XS GIS Cut Line= 3
      3713662.57     10155415.81      3714189.58     10153756.86
      3714137.49     10152840.19
#Sta/Elev= 30
       0   270.2   295.9  262.66     645   257.6   693.4  257.89   795.4   257.1
   827.6  255.33   917.8  255.48  1187.7  251.35  1264.1  252.24  1359.4  250.69
  1450.9  252.52  1483.2  251.98  1520.7  252.07  1547.4  249.07  1617.5  251.98
  1704.8  251.95  1735.8  248.83  1756.5  249.31  1786.5  250.36  1796.5  250.07
  1816.6   245.3  1826.6  245.98  1836.6  250.08  1855.4  251.83  1926.7  252.42
  1956.8  254.35  2217.2  260.62  2427.5  266.62  2627.9   274.1  2658.8  274.22
#Mann= 9 ,-1 , 0
       0     .11       0     645     .17       0   693.4     .11       0
   917.8     .15       0  1483.2     .11       0  1756.5     .17       0
  1786.5     .09       0  1836.6     .15       0  1956.8     .11       0
Bank Sta=1786.5,1836.6
XS Rating Curve= 0 ,0
Exp/Cntr=0.3,0.1

Type RM Length L Ch R = 1 ,51870   ,783,783,783
BEGIN DESCRIPTION:
LITTLE CANEY CREEK 61.0
END DESCRIPTION:
XS GIS Cut Line= 4
      3713720.91     10155364.76      3714246.87     10154163.11
      3714710.41     10153590.19      3714689.58     10152621.44
#Sta/Elev= 30
       0  269.18   440.7  259.09   507.6  259.45     659  256.66  1107.1  256.12
  1215.7  253.17  1247.4  250.67  1370.6  251.93  1527.2  250.88    1556  249.61
  1562.4  246.93  1570.4  246.21  1584.5  250.24  1597.6  251.67  1739.9  250.53
  1776.6  252.53  1797.4   252.6  1875.8  251.66  2024.5  252.35  2097.8  249.89
  2127.8  251.88  2147.8  244.21  2177.8  251.86  2257.8  251.12  2347.9  252.94
  2477.9  258.69  2557.9  260.27  2677.9  266.48  2707.9  266.32  3017.6  276.69
#Mann= 8 ,-1 , 0
       0     .11       0   440.7     .17       0     659     .15       0
  1776.6     .15       0  1797.4     .11       0  1875.8     .17       0
  2127.8     .09       0  2177.8     .17       0
Bank Sta=2127.8,2177.8
XS Rating Curve= 0 ,0
Exp/Cntr=0.3,0.1

Type RM Length L Ch R = 1 ,51087   ,1605,1605,1605
BEGIN DESCRIPTION:
LITTLE CANEY CREEK 60.0
END DESCRIPTION:
XS GIS Cut Line= 5
      3713918.74     10155069.38      3714309.37     10154168.32
      3714726.04     10153621.44      3715423.95     10153564.15
      3715226.21     10152304.86
#Sta/Elev= 30
    2481  261.02  2806.1   256.6  2890.5  257.58  3165.7  256.29  3293.5  255.04
  3383.8  249.74  3637.9   251.6  3681.5  246.73  3702.3     250  3731.4   252.1
  3866.5  250.55  3901.9  252.16  4030.7  251.01    4116  252.66  4262.8  250.71
  4804.6  248.55  4965.3  250.34  4975.5  249.87  4988.7  243.59  5002.7  243.59
  5005.8  247.96    5016  250.55  5157.7  249.42  5232.5  252.67  5329.8   260.6
  5389.8   262.1  5504.8  257.35  5623.3  262.71  5685.9  263.67  6125.6  271.91
#Mann= 8 ,-1 , 0
    2481     .11       0  2890.5     .17       0  3165.7     .15       0
  4965.3     .09       0    5016     .15       0  5232.5     .11       0
  5389.8     .17       0  5685.9     .11       0
Bank Sta=4965.3,5016
XS Rating Curve= 0 ,0
Exp/Cntr=0.3,0.1

Type RM Length L Ch R = 1 ,49482   ,395,395,395
BEGIN DESCRIPTION:
LITTLE CANEY CREEK 58.0
END DESCRIPTION:
XS GIS Cut Line= 3
      3716835.41     10154350.58      3716701.24     10153513.57
      3715637.46     10152652.67
#Sta/Elev= 30
  4152.3  265.58  4334.1  263.38    4405   264.5  4415.1  263.69  4420.7  261.49
  4448.4  259.61  4487.7  256.54    4700  250.31  4810.1  247.03  4982.3  248.66
  4988.6  246.18  4991.3  240.98  5006.2  240.98  5017.8  247.07  5025.7  248.35
  5054.5   246.9  5060.9  248.09  5068.7     247  5184.8  247.13  5348.9  248.68
  5423.8  251.06  5512.5  250.66  5537.4  249.81  5650.9  251.88  5793.2  257.16
  5914.7  256.12  6156.1  258.78  6234.4  259.86  6347.9  264.47  6368.5  263.58
#Mann= 8 ,-1 , 0
  4152.3     .17       0  4448.4     .11       0    4700     .15       0
  4982.3     .09       0  5025.7     .15       0  5184.8     .11       0
  5348.9     .15       0  5512.5     .11       0
Bank Sta=4982.3,5025.7
XS Rating Curve= 0 ,0
Exp/Cntr=0.3,0.1

Type RM Length L Ch R = 1 ,49087   ,697,697,697
BEGIN DESCRIPTION:
LITTLE CANEY CREEK 57.0
END DESCRIPTION:
XS GIS Cut Line= 3
       3717835.4     10154355.81      3716939.58     10153277.69
      3715713.25      10152565.8
#Sta/Elev= 30
  3599.3  269.13  3683.4  266.67  3896.1  261.23  3983.9  260.87  4082.2   254.9
  4154.5  250.15  4218.3  251.01  4403.2  248.25  4464.5  248.56    4730  247.23
  4779.5  246.28  4808.1  243.34  4865.4  247.48  4886.2  247.91  4907.1  244.58
  4921.4   246.7  4970.9  247.61  4978.7  245.81  4985.4  240.71  5000.7  240.71
  5014.6  246.42  5022.3  247.55  5225.9  246.56  5327.8  248.99  5600.9  249.75
  5937.1  255.29    6009  254.39    6125   256.3  6183.8  255.49    6419  261.22
#Mann= 8 ,-1 , 0
  3599.3     .17       0  3683.4     .11       0  3896.1     .17       0
  4082.2     .11       0  4464.5     .15       0  4970.9     .09       0
  5022.3     .15       0  5600.9     .11       0
Bank Sta=4970.9,5022.3
XS Rating Curve= 0 ,0
Exp/Cntr=0.3,0.1

Type RM Length L Ch R = 1 ,48390   ,650,650,650
BEGIN DESCRIPTION:
LITTLE CANEY CREEK 56.0
END DESCRIPTION:
XS GIS Cut Line= 3
      3718017.83     10154461.03      3717343.79     10152910.51
      3715917.83     10151461.05
#Sta/Elev= 30
  3309.3   274.7  3451.8  268.56  3592.5  266.45  3865.2  254.73  3984.9  250.98
  4070.7  248.31  4175.4  250.32  4279.7  248.96  4496.5  247.55  4519.6  245.75
    4814   247.4  4823.1  247.02  4846.6  241.03  4868.5  241.45  4880.9  245.28
  4904.4  248.06  4988.5  248.49  4995.9  240.39  5011.6  240.39  5025.1  248.54
  5109.9  246.23  5279.6  247.95  5392.5  252.43  5484.7  258.03  5555.4  259.37
  6000.8     253    6396  259.12    6609  261.16  6913.6  267.79  7033.3  272.13
#Mann= 9 ,-1 , 0
  3309.3     .11       0  3865.2     .17       0  3984.9     .11       0
  4279.7     .15       0  4988.5     .09       0  5025.1     .15       0
  5392.5     .11       0    6396     .17       0  6913.6     .11       0
Bank Sta=4988.5,5025.1
XS Rating Curve= 0 ,0
Exp/Cntr=0.3,0.1

Type RM Length L Ch R = 1 ,47740   ,448,448,448
BEGIN DESCRIPTION:
LITTLE CANEY CREEK 55.0
END DESCRIPTION:
XS GIS Cut Line= 3
      3718179.15     10154350.59       3717705.2      10152532.9
      3717017.72     10151168.36
#Sta/Elev= 30
  3115.3   272.5  3419.5  260.96  3580.6   257.6    3669  252.91  3703.2  251.25
  3793.7  248.03  3853.7  245.93  4034.6  247.14    4051  245.53  4675.3  246.43
    4721  239.53  4736.8  239.53  4747.6  247.07    4975  248.76  4992.1  241.65
  5000.2  241.21  5016.9  248.03  5029.4  248.69  5128.5   246.7  5150.8  244.03
    5201   248.5  5312.5  246.21  5433.2  247.44  5535.6  248.67  5580.3  245.73
  5589.3  247.86  5678.9  251.38  5730.8  250.46  6037.2  257.73  6521.7  264.52
#Mann= 8 ,-1 , 0
  3115.3     .17       0  3419.5     .11       0    3669     .17       0
  3703.2     .11       0  3793.7     .15       0  4675.3     .09       0
  4747.6     .15       0  5433.2     .11       0
Bank Sta=4675.3,4747.6
XS Rating Curve= 0 ,0
Exp/Cntr=0.3,0.1

Type RM Length L Ch R = 1 ,47292   ,599,599,599
BEGIN DESCRIPTION:
LITTLE CANEY CREEK 54.0
END DESCRIPTION:
XS GIS Cut Line= 3
      3718538.53     10154225.57      3717994.82     10152265.59
      3717892.78     10151231.61
#Sta/Elev= 30
    2966  273.64  3608.9  252.28  3734.4  244.58  3790.5   245.7  3881.9  242.56
  3894.3  245.49  3921.3  242.36  3926.5  244.19  3955.6  242.86  3960.8  245.27
  3995.1  242.29  4091.5  242.45  4147.7  245.66    4216  242.19  4300.4   244.9
  4368.9  242.57  4408.4   245.2  4527.3  245.61    4669  242.64  4880.2  247.36
  4983.9  246.94  5006.6  239.46  5022.6  239.46  5024.8  247.21  5084.9  245.64
  5222.1  254.49    5336  257.86  5456.7  260.58  5898.9  259.47    6039  263.23
#Mann= 5 ,-1 , 0
    2966     .11       0  3608.9     .15       0  4983.9     .09       0
  5024.8     .15       0    5336     .11       0
Bank Sta=4983.9,5024.8
XS Rating Curve= 0 ,0
Exp/Cntr=0.3,0.1

Type RM Length L Ch R = 1 ,46693   ,674,674,674
BEGIN DESCRIPTION:
LITTLE CANEY CREEK 53.0
END DESCRIPTION:
XS GIS Cut Line= 3
      3718767.85     10154461.07       3718371.8     10152237.16
      3718095.82     10151048.48
#Sta/Elev= 30
  2741.1  287.94    2863  286.56  3005.2  277.59  3127.1  272.93  3421.6  266.68
  3502.9  262.53  3553.7  255.65  3620.7  250.49  3817.8  245.23  3848.2  242.35
  3878.7  244.14  3919.4  241.32  3949.8  246.53  4363.9  244.03  4772.6  244.12
  4965.6  246.66  4975.7  245.67  4984.5  239.02  5000.5  239.02  5016.5  247.18
    5191  244.68  5216.6  247.39  5232.1  252.45  5259.2  256.38  5323.5  258.81
  5416.9  260.93  5482.7  258.02  5673.5  260.56  6022.6  259.72  6220.3   263.6
#Mann= 5 ,-1 , 0
  2741.1     .11       0  3620.7     .15       0  4965.6     .09       0
  5016.5     .15       0  5323.5     .11       0
Bank Sta=4965.6,5016.5
XS Rating Curve= 0 ,0
Exp/Cntr=0.3,0.1

Type RM Length L Ch R = 1 ,46019   ,830,830,830
BEGIN DESCRIPTION:
LITTLE CANEY CREEK 52.0
END DESCRIPTION:
XS GIS Cut Line= 3
      3719006.42      10154204.8      3718884.89     10152216.93
      3718555.04     10151127.56
#Sta/Elev= 30
  2998.9   280.2  3112.8  279.69  3303.2  268.02  3533.6  258.35  3548.8  256.39
  3580.7  256.53  3582.6  256.48  3789.2  247.75    3878  245.48  3894.3  244.37
  3915.9   239.8  3932.9   239.8  3934.4  242.65  3954.4  245.45  3994.5  243.54
  4084.7  245.22  4605.6  243.12  4705.8  244.39  4745.9  247.37  4906.2   241.3
  4976.3  245.33  4990.5  242.58  4994.4     240  5017.5  244.78  5103.7  244.71
  5334.6   257.4  5613.1  258.91  5748.9  256.99  5853.4  260.51  6128.7  260.31
#Mann= 7 ,-1 , 0
  2998.9     .11       0  3580.7     .15       0  3582.6     .11       0
  3789.2     .15       0  4976.3     .09       0  5017.5     .15       0
  5334.6     .11       0
Bank Sta=4976.3,5017.5
XS Rating Curve= 0 ,0
Exp/Cntr=0.3,0.1

Type RM Length L Ch R = 1 ,45189   ,1177,1177,1177
BEGIN DESCRIPTION:
LITTLE CANEY CREEK 51.0
END DESCRIPTION:
XS GIS Cut Line= 4
      3719978.63     10153510.33      3719386.66     10153163.35
      3719219.09     10151982.56      3719019.44     10151700.44
#Sta/Elev= 30
  3125.8  281.44  3184.7  279.55  3242.6  272.38  3346.4  266.23  3502.7  253.25
  3592.6  248.63    3624  249.68  3651.2  247.04  3694.7  249.56  3945.6  244.12
    4199  243.23  4228.4  240.37    4270  243.17  4460.7   243.9  4501.1  239.64
  4531.4  245.12  4624.7  243.28  4703.1  245.49  4979.3  244.49  4985.9  242.25
    4988  238.51    5004  238.51 5012.85244.7134  5020.1  245.19  5028.7  249.63
  5043.2  252.39  5073.9  253.29  5178.9  255.55  5190.4  255.32  5350.2  257.69
#Mann= 7 ,-1 , 0
  3125.8     .17       0  3502.7     .15       0  4979.3     .09       0
 5012.85     .15       0  5073.9     .17       0  5178.9     .15       0
  5190.4     .11       0
Bank Sta=4979.3,5012.85
XS Rating Curve= 0 ,0
Exp/Cntr=0.3,0.1

Type RM Length L Ch R = 1 ,44017   ,1234,1234,1234
BEGIN DESCRIPTION:
LITTLE CANEY CREEK 50.0
END DESCRIPTION:
XS GIS Cut Line= 3
      3720152.25     10153397.49      3719690.31     10152104.75
      3718731.27     10151422.84
#Sta/Elev= 30
       0   273.1   155.5  270.23     336   257.3   409.7  250.11     415  250.87
   440.4  247.34   563.6  241.94   891.6  242.38   917.1  239.18   941.3  242.21
   978.7  242.72  1196.2  242.87  1214.4  238.44    1228  242.92  1281.3     242
    1391     245    1557  253.35  1598.8  253.85  1678.8  250.87  1800.5  251.43
  1878.9  250.17    2044  252.87  2079.7  254.52  2094.5  256.76  2130.1  256.12
  2144.9  258.22  2216.2  255.78  2367.5  254.74  2417.9  256.95  2548.6   258.7
#Mann= 6 ,-1 , 0
       0     .17       0     415     .15       0  1196.2     .09       0
    1228     .15       0    1557     .17       0  1800.5     .11       0
Bank Sta=1196.2,1228
XS Rating Curve= 0 ,0
Exp/Cntr=0.3,0.1

Type RM Length L Ch R = 1 ,42778   ,1460,1460,1460
BEGIN DESCRIPTION:
LITTLE CANEY CREEK 49.0
END DESCRIPTION:
XS GIS Cut Line= 3
      3721371.88       10152460.      3720482.11      10151761.2
       3718737.3     10151379.25
#Sta/Elev= 30
  3711.2  273.39  4154.9  252.79  4175.7  247.78  4198.2  248.97  4204.6  247.34
    4219  250.85  4239.8  249.13  4275.8  251.53  4283.2  248.52  4318.5  244.32
  4451.4   242.4  4560.7  241.38  4581.5  238.61  4796.5  238.43  4823.7  241.73
  4962.4  241.02    4980  242.46  5003.3  235.25  5019.4  235.25    5021  237.89
  5031.2  241.95  5041.4  242.61  5205.2  240.65    5410  242.47  5573.7  240.89
  5622.7  243.54  5722.9   250.5    6188  249.76    6414  256.43  6628.7  259.24
#Mann= 6 ,-1 , 0
  3711.2     .11       0  4451.4     .15       0    4980     .09       0
  5041.4     .15       0  5622.7     .17       0  5722.9     .11       0
Bank Sta=4980,5041.4
XS Rating Curve= 0 ,0
Exp/Cntr=0.3,0.1

Type RM Length L Ch R = 1 ,41318   ,463,463,463
BEGIN DESCRIPTION:
LITTLE CANEY CREEK 48.0
END DESCRIPTION:
XS GIS Cut Line= 3
      3721415.26     10152212.58      3719806.02     10150808.76
      3719072.15     10150593.85
#Sta/Elev= 30
  2864.5  269.14  3026.7  263.59  3150.7  256.26  3239.4  249.85  3339.4  247.01
  3449.6   242.9  3495.8  242.21  3662.2  241.24  3756.8  242.53  3791.9   238.7
  3877.3  238.04  3905.8  239.86  3948.5  238.04    3976  238.63  3983.6   241.9
  3997.9  243.24  4012.1     240  4075.7  235.44  4096.6  239.86  4188.7  241.65
  4975.7  239.67  4983.3   238.3  4987.4  234.31  5003.6  234.31  5018.9  239.64
  5091.9  241.42  5164.8  246.45  5294.7  247.92  5472.2  254.64  5764.7  256.75
#Mann= 9 ,-1 , 0
  2864.5     .11       0  3150.7     .17       0  3339.4     .11       0
  3449.6     .17       0  3495.8     .11       0  3662.2     .15       0
  4975.7     .09       0  5018.9     .15       0  5294.7     .17       0
Bank Sta=4975.7,5018.9
XS Rating Curve= 0 ,0
Exp/Cntr=0.3,0.1

Type RM Length L Ch R = 1 ,40855   ,690,690,690
BEGIN DESCRIPTION:
LITTLE CANEY CREEK 47.0
END DESCRIPTION:
XS GIS Cut Line= 3
      3721442.15     10152097.11      3719947.39     10150617.97
      3718929.96     10150385.71
#Sta/Elev= 30
  2896.7  268.71  2993.1  265.02  3361.5  245.55  3636.1  240.78  4127.3  240.51
  4148.5  237.67  4155.6  239.76  4162.7  236.79  4169.7   239.6    4191  232.26
    4198  235.87  4205.1  231.63  4212.1   233.8  4231.8  231.15    4249  231.15
  4261.7  238.38  4275.8   240.6  4579.9  239.08  4728.4  241.32  4869.8  237.27
  4940.5  240.06    4990  238.87  5006.2  233.62  5019.6  238.29  5102.4  239.52
  5231.4  250.31  5401.1  249.38  5681.7  256.89  5881.2  253.14  6043.2  256.73
#Mann= 7 ,-1 , 0
  2896.7     .11       0  2993.1     .17       0  3361.5     .11       0
  3636.1     .15       0    4990     .09       0  5019.6     .15       0
  5401.1     .17       0
Bank Sta=4990,5019.6
XS Rating Curve= 0 ,0
Exp/Cntr=0.3,0.1

Type RM Length L Ch R = 1 ,40165   ,528,528,528
BEGIN DESCRIPTION:
LITTLE CANEY CREEK 46.0
END DESCRIPTION:
XS GIS Cut Line= 3
      3721447.36     10151935.65      3719978.64     10150050.26
      3719077.61     10149925.27
#Sta/Elev= 30
  2719.1   267.5  3149.1   245.2  3263.5     241  3357.4  240.78  4260.5  239.76
  4382.7  239.03  4397.1  238.27  4403.5  235.08  4438.8  237.57  4552.8   239.6
  4674.9  239.66  4689.4  238.07  4716.5  240.42  4753.1  238.22  4809.7  239.65
  4838.7  237.92  4944.5  238.97  4967.1  236.43  4973.5  237.25  4986.2  232.08
  5002.4  232.08  5008.7  233.52  5016.9  238.21  5023.2  234.87  5031.4  237.98
  5037.7  237.31  5044.6  239.35  5280.8  240.29  5542.2  249.82  6018.7   257.5
#Mann= 6 ,-1 , 0
  2719.1     .17       0  3149.1     .11       0  3357.4     .15       0
  4944.5     .09       0  5044.6     .15       0  5542.2     .17       0
Bank Sta=4944.5,5044.6
XS Rating Curve= 0 ,0
Exp/Cntr=0.3,0.1

Type RM Length L Ch R = 1 ,39637   ,1000,1000,1000
BEGIN DESCRIPTION:
LITTLE CANEY CREEK 45.0
END DESCRIPTION:
XS GIS Cut Line= 4
      3721483.88     10151878.42      3720525.52     10150649.22
      3720317.18     10149987.76        3719213.     10149852.34
#Sta/Elev= 30
    2596  267.77  2666.9  265.11  2940.3  248.99  3053.9  244.73    3065  244.57
  3118.5  241.92  3232.5  240.96  3873.3  240.13  3980.6  238.01  4001.4  239.61
  4341.4  238.69  4351.9   238.3  4365.4  234.12  4397.8  239.08  4430.2  237.13
  4887.8  239.87  4988.5  238.03  4998.6     235  5000.6  231.52  5016.8  231.52
  5025.1  236.13  5030.1  234.42    5049  238.29  5089.3  240.14  5300.8  241.53
    5602  250.42  5713.9  251.59  5824.7   248.4  5848.9  250.55  5960.6  252.54
#Mann= 7 ,-1 , 0
    2596     .11       0  2666.9     .17       0  3053.9     .11       0
    3065     .15       0  4988.5     .09       0    5049     .15       0
    5602     .17       0
Bank Sta=4988.5,5049
XS Rating Curve= 0 ,0
Exp/Cntr=0.3,0.1

Type RM Length L Ch R = 1 ,38637   ,1059,1059,1059
BEGIN DESCRIPTION:
LITTLE CANEY CREEK 44.0
END DESCRIPTION:
XS GIS Cut Line= 5
      3721499.48     10151836.74      3720556.77     10150649.22
      3720425.31     10149624.43      3720226.24     10149426.26
      3719573.12      10148665.7
#Sta/Elev= 30
  2169.7  267.26  2321.1  260.75  2502.3  249.24  2658.2  242.77  3420.3  240.07
  3542.1  237.33  3577.3  239.34  3845.4  238.31  3865.5  235.78  3905.9  239.18
  3951.8  233.99  3976.4  238.54  4016.8  239.07  4663.4  238.43  4718.3  237.42
  4726.8  235.23  4797.5  237.85  4889.4  235.66    4946  237.81  4967.2  234.85
  4980.2  229.86  5023.6  233.09  5031.3  236.75  5045.5   238.2  5468.8  240.49
  5584.3  242.85  5598.6  246.29  5626.4  244.02  5818.1  256.05  6002.5  263.41
#Mann= 6 ,-1 , 0
  2169.7     .11       0  2321.1     .17       0  2658.2     .15       0
    4946     .09       0  5045.5     .15       0  5468.8     .17       0
Bank Sta=4946,5045.5
XS Rating Curve= 0 ,0
Exp/Cntr=0.3,0.1

Type RM Length L Ch R = 1 ,37578   ,503,503,503
BEGIN DESCRIPTION:
LITTLE CANEY CREEK 43.0
END DESCRIPTION:
XS GIS Cut Line= 3
      3722108.89     10150013.83      3720546.35     10149138.81
      3719667.88     10148411.09
#Sta/Elev= 30
  3499.3  256.91  3613.4  254.06    3624  254.43  3855.8  253.54  3962.5  250.64
  4148.8  246.31  4213.9  247.28  4370.3  240.42  4516.4  236.54  4656.8  237.71
  4737.9  234.52  4781.3  234.88  4808.7  237.87  4840.6  235.72  4911.4  235.08
    4965  237.29  4986.7  235.09    4993  230.36  5010.9  230.36  5024.4  235.36
  5251.6  238.36  5337.6   235.5  5387.1  237.13  5436.5  235.78  5450.9  237.37
  5755.7   236.7  5842.2  241.78  5954.9  251.71  6082.5  253.62  6430.9  271.97
#Mann= 7 ,-1 , 0
  3499.3     .17       0  3613.4     .11       0    3624     .17       0
  3962.5     .15       0  4986.7     .09       0  5024.4     .15       0
  5842.2     .17       0
Bank Sta=4986.7,5024.4
XS Rating Curve= 0 ,0
Exp/Cntr=0.3,0.1

Type RM Length L Ch R = 1 ,37075   ,509,509,509
BEGIN DESCRIPTION:
LITTLE CANEY CREEK 42.0
END DESCRIPTION:
XS GIS Cut Line= 3
      3722051.52     10149940.86      3720681.77     10148784.64
      3719723.46      10148310.7
#Sta/Elev= 30
  3306.7  255.17  3669.5     254  3728.2  251.91  3923.5  249.34  3997.4  247.68
  4046.8  248.55  4094.2   246.3  4139.1  243.34  4245.7  242.13  4317.2  235.21
  4352.3  237.33  4473.2  236.46  4529.2  235.67  4572.1  233.13  4586.4  235.46
  4707.3  237.46  4777.6  236.94  4813.9   233.1  4842.5  232.72  4869.9  232.96
  4906.2  235.93  4976.5  236.29  4984.2  235.66  4996.1  228.47    5014  228.47
  5019.4  236.75  5449.4  236.48  5595.3  242.26  5873.3   257.8  6168.3  269.46
#Mann= 7 ,-1 , 0
  3306.7     .17       0  3669.5     .15       0  3923.5     .11       0
  4094.2     .15       0  4976.5     .09       0  5019.4     .15       0
  5595.3     .17       0
Bank Sta=4976.5,5019.4
XS Rating Curve= 0 ,0
Exp/Cntr=0.3,0.1

Type RM Length L Ch R = 1 ,36566   ,1076,1076,1076
BEGIN DESCRIPTION:
LITTLE CANEY CREEK 41.0
END DESCRIPTION:
XS GIS Cut Line= 3
      3722088.02     10149904.44      3720832.81     10148519.01
      3719785.94     10148201.31
#Sta/Elev= 30
  3286.6  255.83  3423.8   253.6  3480.1  254.97  3660.2  253.58  3938.2   245.8
  4013.7  243.09  4038.4  244.63  4067.9   244.7  4110.5  240.85  4209.1  239.83
  4273.4   235.1  4287.6  236.49  4343.7  234.42  4450.4  234.19  4492.3  235.78
  4599.1  234.65  4620.1  230.83    4641  234.34    4712  236.25    4981  234.75
  4988.4  232.42  4993.7  227.59  5011.6  227.59  5016.8  232.34  5023.5  235.08
  5143.8  236.98  5374.2  235.36    5651  238.73  6096.3  261.96  6250.1  265.93
#Mann= 8 ,-1 , 0
  3286.6     .17       0  3660.2     .15       0  3938.2     .11       0
  4013.7     .17       0  4038.4     .15       0    4981     .09       0
  5023.5     .15       0    5651     .17       0
Bank Sta=4981,5023.5
XS Rating Curve= 0 ,0
Exp/Cntr=0.3,0.1

Type RM Length L Ch R = 1 ,35490   ,574,574,574
BEGIN DESCRIPTION:
LITTLE CANEY CREEK 40.0
END DESCRIPTION:
XS GIS Cut Line= 3
      3722108.86     10149222.15      3721419.55       10148582.
      3720198.48     10147395.07
#Sta/Elev= 30
  4297.1  252.63  4631.1  245.84    4709  240.74  4772.8  235.78  4801.1  237.03
  4815.3  234.12  4843.7  235.35  4850.5  237.74  4885.6  237.99    4914  237.14
  4949.7  231.61  4963.8  234.61    4978  235.36  4984.8  234.28  4990.1  229.53
    5008  229.53  5041.5  235.58    5105  233.56  5140.7  235.51  5183.2  233.34
  5317.5  236.99  6010.4  235.69  6045.9   234.5  6081.2   235.9  6328.6  236.67
  6392.4  237.98  6493.5  243.36  6646.6  253.25  6809.2  260.88  6940.7  266.85
#Mann= 7 ,-1 , 0
  4297.1     .17       0    4709     .15       0    4978     .09       0
  5041.5     .15       0  6493.5     .11       0  6646.6     .15       0
  6809.2     .11       0
Bank Sta=4978,5041.5
XS Rating Curve= 0 ,0
Exp/Cntr=0.3,0.1

Type RM Length L Ch R = 1 ,34916   ,490,490,490
BEGIN DESCRIPTION:
LITTLE CANEY CREEK 39.0
END DESCRIPTION:
XS GIS Cut Line= 3
      3722874.51     10149045.07      3721557.92     10148444.48
      3720117.83     10147011.05
#Sta/Elev= 30
  3552.9   255.1  3840.1  256.24  4179.1  251.94  4225.2  250.59  4271.2  245.67
  4380.9  241.94  4541.2  235.95  4626.4  236.88  4661.8  235.54  4684.9  231.65
  4725.3  234.08  4736.5  231.36    4754  231.44  4782.5  236.55  4828.6  234.54
  4835.2  229.71  4846.2  229.72  4868.2  234.93  4966.8  233.33  4972.3  233.93
  4986.4  226.88  5004.4  226.88  5023.7  232.98  5094.4  236.93  5999.5  235.33
  6183.3  236.63  6284.9  239.93  6664.2  262.31  6939.9  282.86  7031.9  292.35
#Mann= 6 ,-1 , 0
  3552.9     .17       0  4380.9     .15       0  4966.8     .12       0
  4972.3     .09       0  5023.7     .15       0  6284.9     .11       0
Bank Sta=4972.3,5023.7
XS Rating Curve= 0 ,0
Exp/Cntr=0.3,0.1

Type RM Length L Ch R = 1 ,34426   ,268,268,268
BEGIN DESCRIPTION:
LITTLE CANEY CREEK 38.0
END DESCRIPTION:
XS GIS Cut Line= 3
      3722367.87     10148761.09      3721758.52     10148186.55
      3720338.03      10146940.9
#Sta/Elev= 30
  4162.5  253.03  4212.1  252.79  4268.7   250.2  4360.6  244.59  4390.2  241.05
  4417.2  238.11  4494.9  235.98  4643.6  235.03  4869.9  236.77  4926.6  235.75
  4969.1  232.23  4975.9  230.76  4981.1  226.94  4999.1  226.94  5011.7  232.56
  5046.8  232.84  5067.7  230.88  5089.5   232.3  5146.5  230.34  5188.2  235.31
  5238.5  236.42  5280.3  235.03  5479.6  235.99  5500.4  234.84  5911.4  234.61
  6230.2  236.68  6325.9  239.14  6394.9  241.85    6427  243.27  6889.3  271.71
#Mann= 7 ,-1 , 0
  4162.5     .17       0  4390.2     .15       0  4969.1     .09       0
  5011.7     .15       0  6325.9     .11       0  6394.9     .15       0
    6427     .11       0
Bank Sta=4969.1,5011.7
XS Rating Curve= 0 ,0
Exp/Cntr=0.3,0.1

Type RM Length L Ch R = 1 ,34158   ,726,726,726
BEGIN DESCRIPTION:
LITTLE CANEY CREEK 37.0
END DESCRIPTION:
XS GIS Cut Line= 3
      3722655.72     10148617.97      3721936.97     10147987.76
      3720983.84     10146722.13
#Sta/Elev= 30
  4051.3  254.92  4068.9  255.61  4160.9  251.87  4175.2  252.47  4288.1  244.39
  4330.8  242.83  4373.5  237.89  4407.3   236.4  4473.1  234.18  4806.2  235.56
  4819.8  235.07    4848  229.83  4855.6  229.77  4898.3  234.74  4976.1  235.77
  4982.8  234.72  4990.3  229.96  5002.7  225.19  5020.7  225.19  5047.1  232.93
  5082.5  235.92  5617.6  233.81  5996.6  234.55    6248  240.49  6396.3  244.36
  6425.5   246.6  6460.9  246.22    6540  250.74  6560.8  249.47  6591.6  252.11
#Mann= 5 ,-1 , 0
  4051.3     .17       0  4407.3     .15       0  4976.1     .09       0
  5082.5     .15       0    6248     .11       0
Bank Sta=4976.1,5082.5
XS Rating Curve= 0 ,0
Exp/Cntr=0.3,0.1

Type RM Length L Ch R = 1 ,33432   ,499,499,499
BEGIN DESCRIPTION:
LITTLE CANEY CREEK 36.0
END DESCRIPTION:
XS GIS Cut Line= 3
      3723322.41     10148451.32      3722154.27     10147509.87
      3721151.65     10146613.78
#Sta/Elev= 30
  3499.7  252.81  3569.1   250.6    3729  242.28  3794.7  239.88  4085.8  237.67
  4277.8  234.31  4762.4  235.42    4812  231.86  4840.8  231.93  4861.6  229.21
  4890.4  233.17  4911.2  229.94  4925.6  232.65    4932  231.19    4940  233.14
  4960.8  233.54  4968.7  230.05  4973.6  225.51  4991.6  225.51  5003.8  230.43
  5024.7  233.61  5053.1  235.67  5095.8  232.06  5130.9  231.37  5209.4  235.01
  5711.9  233.65    5884  241.18  6064.4  247.93  6256.2  253.85  6344.7  256.79
#Mann= 8 ,-1 , 0
  3499.7     .11       0  3569.1     .17       0    3729     .15       0
  4960.8     .09       0  5024.7     .15       0    5884     .17       0
  6064.4     .15       0  6256.2     .11       0
Bank Sta=4960.8,5024.7
XS Rating Curve= 0 ,0
Exp/Cntr=0.3,0.1

Type RM Length L Ch R = 1 ,32933   ,502,502,502
BEGIN DESCRIPTION:
LITTLE CANEY CREEK 35.0
END DESCRIPTION:
XS GIS Cut Line= 3
      3723367.84     10148311.05      3722271.94     10147092.98
      3721535.95     10146367.99
#Sta/Elev= 30
  3361.5  251.99  3454.7  248.75  3666.1  238.67  3857.5  236.15  3879.7  236.07
  4062.2  235.51  4182.5  232.99  4345.5  233.97  4373.9  231.53  4388.1  233.38
  4444.9  234.74  4883.6  234.94  4905.3  233.03  4975.7  234.73    4983  232.62
  4988.2  223.75  5006.2  223.75  5025.4   234.2  5188.1  233.38  5230.5  230.18
  5258.8  229.92  5315.3  232.92  5414.3  232.09  5566.2  236.76  5628.3  239.57
  5746.8  245.09  5832.6  246.81  5951.8  249.99  6008.4  254.19  6033.1  254.42
#Mann= 9 ,-1 , 0
  3361.5     .11       0  3454.7     .17       0  3857.5     .11       0
  3879.7     .15       0  4975.7     .09       0  5025.4     .15       0
  5566.2     .11       0  5628.3     .15       0  5832.6     .11       0
Bank Sta=4975.7,5025.4
XS Rating Curve= 0 ,0
Exp/Cntr=0.3,0.1

Type RM Length L Ch R = 1 ,32431   ,1123,1123,1123
BEGIN DESCRIPTION:
LITTLE CANEY CREEK 34.0
END DESCRIPTION:
XS GIS Cut Line= 3
      3723417.83     10148111.04      3722541.14     10146722.14
      3721717.85     10146011.07
#Sta/Elev= 30
  3563.5  250.71  3678.6  245.87  3843.4   238.4  3962.9  233.99  4228.7  233.38
  4345.4  231.84  4433.6  233.21  4470.1  230.17  4485.4  232.19  4543.1  233.41
  4956.1   234.5  4974.2   224.7  4992.2   224.7  4998.5  229.84  5019.7  234.06
  5150.3  233.13    5202  230.42  5244.6  234.03  5322.5  231.39  5343.3  232.99
  5379.5   230.4  5414.6   232.6  5500.1  233.37  5535.3  231.55  5570.4  232.75
  5598.9  231.25  5820.2  236.54  5989.3   241.7  6145.2  247.73  6293.8  257.59
#Mann= 8 ,-1 , 0
  3563.5     .11       0  3678.6     .17       0  3843.4     .11       0
  4228.7     .15       0  4956.1     .09       0  5019.7     .15       0
  5820.2     .17       0  5989.3     .11       0
Bank Sta=4956.1,5019.7
XS Rating Curve= 0 ,0
Exp/Cntr=0.3,0.1

Type RM Length L Ch R = 1 ,31308   ,966,966,966
BEGIN DESCRIPTION:
Mapping XS 043cb405
END DESCRIPTION:
XS GIS Cut Line= 3
      3723588.04     10147899.27      3722942.18      10146508.6
       3721771.6     10145868.68
#Sta/Elev= 30
  4034.6  248.21  4309.1  235.64  4395.5  235.21  4412.6  235.37  4953.8  231.99
  4980.8  231.97  4991.4  229.64  4993.8  224.98    5012  224.98  5019.9  232.03
  5277.2  230.49  5499.8  234.68  5575.9  233.41  5607.1  227.99  5673.6  228.97
  5679.3  232.03  5695.4   228.8  5701.1  231.74    5835  227.18  5864.3  233.49
  5880.4  232.15  5886.1  226.47  5907.9  232.88  5945.8  233.98    6202  229.46
  6304.9   235.7  6319.5  236.58  6597.9  246.13  6761.3  252.75    6902   260.1
#Mann= 11 ,-1 , 0
  4034.6     .17       0  4309.1     .11       0  4395.5     .17       0
  4412.6     .11       0  4953.8     .15       0  4980.8     .09       0
  5019.9     .15       0  6304.9     .17       0  6319.5     .11       0
  6597.9     .17       0  6761.3     .11       0
Bank Sta=4980.8,5019.9
XS Rating Curve= 0 ,0
Exp/Cntr=0.3,0.1

Type RM Length L Ch R = 1 ,30342   ,569,569,569
BEGIN DESCRIPTION:
LITTLE CANEY CREEK 33.0
END DESCRIPTION:
XS GIS Cut Line= 3
      3723806.77     10147341.98      3723713.02     10146649.22
      3721867.85     10145911.07
#Sta/Elev= 30
  4570.3  243.79  4898.5  241.53  4964.8  235.37  4971.1  232.57  4976.1  233.11
 4983.51230.0795    4995  227.36    4996  225.66  5014.3  225.66  5014.8  226.16
  5015.2  228.58  5025.3   230.1  5176.7  231.25  5227.1  227.97  5263.7  233.87
  5381.4  232.66  5981.7  233.02    6488   232.5  6524.3  229.34  6541.9  232.28
  6571.5  232.35  6619.9  230.39    6632  228.42  6654.9  231.81  6708.8  232.86
  6763.4   237.7  6870.3  243.67  7063.3  247.36  7232.8  253.32  7256.7  254.71
#Mann= 8 ,-1 , 0
  4570.3     .11       0 4983.51     .06       0  5025.3     .11       0
  5263.7     .11       0  5981.7     .15       0  6763.4     .11       0
  7063.3     .17       0  7232.8     .11       0
Bank Sta=4983.51,5025.3
XS Rating Curve= 0 ,0
Exp/Cntr=0.3,0.1
