HEC-RAS study CRYSTAL CREEK.prj: CRYSTAL CREEK Base Level Engineering

--- CRYSTAL CREEK.g01 (geometry) --- (continued)

Type RM Length L Ch R = 1 ,54500   ,500,500,500
BEGIN DESCRIPTION:
CRYSTAL CREEK 108.0
END DESCRIPTION:
XS GIS Cut Line= 3
      3867961.24     10111698.43       3867096.6     10111659.73
      3866236.89      10111553.9
#Sta/Elev= 30
  4134.5  183.04  4358.1  170.21  4448.2  166.95  4518.3   167.3  4568.3  169.27
  4728.5  165.99  4855.8  166.19  4918.7  162.91  4948.7  162.94  4958.7  160.43
  4968.7  160.65  4978.7  159.44  4988.7  154.55  4991.5  152.06  5026.1  152.06
    5032  159.07    5039  163.08  5079.3  164.28  5108.1  162.66  5180.1  162.84
  5220.4  159.39  5290.9  161.43  5311.1  159.08  5361.9  163.22  5403.8  161.47
  5502.5  165.94  5600.6  174.89  5605.6  174.31  5643.6     177  5866.2  178.35
#Mann= 4 ,-1 , 0
  4134.5     .17       0  4948.7     .09       0    5039     .15       0
  5403.8     .17       0
Bank Sta=4948.7,5039
XS Rating Curve= 0 ,0
Exp/Cntr=0.3,0.1

Type RM Length L Ch R = 1 ,54000   ,438,438,438
BEGIN DESCRIPTION:
CRYSTAL CREEK 107.0
END DESCRIPTION:
XS GIS Cut Line= 3
      3867998.99     10111579.92      3867248.39     10111247.31
      3866446.87     10110845.27
#Sta/Elev= 30
    4179   184.9  4420.9  170.83  4511.6  166.83  4703.3  167.45  4855.8  162.47
  4913.1  163.93    4958   163.2  4967.8  162.36  4981.3  158.24  4987.2  152.02
  5021.8  152.02  5026.8  158.72  5049.2  163.57  5132.9  162.46  5183.2  157.99
  5222.3  158.64  5227.9   157.5  5244.6  159.82  5278.9  161.47  5317.2  158.81
  5339.6     161  5384.2  160.14  5423.3   165.2  5436.9  169.64  5490.3  174.12
  5638.3  171.05  5817.3  179.09  5839.7  178.64  5875.7  180.55  5896.7  179.68
#Mann= 5 ,-1 , 0
    4179     .17       0  4855.8     .15       0    4958     .09       0
  5049.2     .15       0  5278.9     .17       0
Bank Sta=4958,5049.2
XS Rating Curve= 0 ,0
Exp/Cntr=0.3,0.1

Type RM Length L Ch R = 1 ,53562   ,562,562,562
BEGIN DESCRIPTION:
CRYSTAL CREEK 106.0
END DESCRIPTION:
XS GIS Cut Line= 3
      3868025.04     10111430.35      3867470.58     10110887.72
      3866596.24     10110682.97
#Sta/Elev= 30
  4224.2  182.93  4504.5  168.38  4614.3     167  4688.4   166.8  4810.7  161.45
  4811.5  161.38  4836.8  161.07    4844  158.98    4851  159.81  4858.1  157.93
  4865.1  158.76  4872.3  157.35  4914.7  159.68  4921.7  158.57    4943  158.59
  4971.3  160.91  4985.4  156.72  4990.2  151.74  5024.9  151.74  5033.6   157.2
    5050  161.41  5064.4  162.18  5105.5  160.47    5135  162.08  5182.6  162.19
  5259.6  158.79  5277.7  159.94  5516.3  165.59  5721.7  176.88    5898  173.36
#Mann= 7 ,-1 , 0
  4224.2     .17       0  4614.3     .15       0  4810.7     .17       0
  4811.5     .15       0  4971.3     .09       0    5050     .15       0
  5277.7     .17       0
Bank Sta=4971.3,5050
XS Rating Curve= 0 ,0
Exp/Cntr=0.3,0.1

Type RM Length L Ch R = 1 ,53000   ,486,486,486
BEGIN DESCRIPTION:
CRYSTAL CREEK 105.0
END DESCRIPTION:
XS GIS Cut Line= 3
      3868163.92     10111117.84      3867499.38     10110574.01
      3866563.29     10109799.44
#Sta/Elev= 30
  4141.3  176.77  4392.5  168.63  4555.4  161.19  4590.6  160.54    4648  162.09
  4683.2   159.7  4704.8  161.95  4732.7  162.25  4825.3  161.16  4860.5  162.24
  4882.7  160.44  4932.2  161.18  4946.6  159.28  4975.3  158.57  4989.1  156.44
  4993.1  150.41  5027.9  150.41  5031.3  155.81  5045.6   161.3  5136.3  157.38
  5158.9  162.61  5216.3  165.15  5287.5  163.19  5329.6  163.78  5365.4  161.39
  5586.1  165.49  5969.1  163.73  6104.6  169.97  6174.9  174.65    6215  175.59
#Mann= 4 ,-1 , 0
  4141.3     .17       0  4932.2     .09       0  5045.6     .15       0
  5136.3     .17       0
Bank Sta=4932.2,5045.6
XS Rating Curve= 0 ,0
Exp/Cntr=0.3,0.1

Type RM Length L Ch R = 1 ,52514   ,514,514,514
BEGIN DESCRIPTION:
CRYSTAL CREEK 104.0
END DESCRIPTION:
XS GIS Cut Line= 3
      3868346.26     10110879.17      3867885.34     10110366.91
      3866919.55      10109625.1
#Sta/Elev= 30
  4310.9  173.25  4390.1  170.91  4485.2  168.45  4547.1  170.58  4832.8  160.15
  4860.4  158.15  4896.3  159.16  4910.5  156.23  4931.4   157.4  4945.6  154.93
  4949.9  149.09    5000  149.81  5002.3  154.86  5016.8  152.66  5023.1  155.89
  5045.8  155.64  5052.1  158.18  5072.9  160.33  5101.9  158.55  5116.4 160.722
  5154.7  161.17  5373.9  160.29    5430  157.44  5450.8  161.12  5494.4  159.31
  5558.7  162.03  5652.1  160.94    5808  165.49  6015.5  164.24  6217.8  173.24
#Mann= 6 ,-1 , 0
  4310.9     .17       0  4390.1     .15       0  4547.1     .17       0
  4832.8     .09       0  5116.4     .15       0  5154.7     .17       0
Bank Sta=4832.8,5116.4
XS Rating Curve= 0 ,0
Exp/Cntr=0.3,0.1

Type RM Length L Ch R = 1 ,52000   ,500,500,500
BEGIN DESCRIPTION:
CRYSTAL CREEK 103.0
END DESCRIPTION:
XS GIS Cut Line= 3
       3868511.2     10110215.11      3868098.13     10110026.72
      3867117.83     10109461.06
#Sta/Elev= 30
    4546  175.19  4641.6  175.37  4744.7  171.74  4894.3  163.46  4913.2  162.61
  4929.1  159.01  4957.6   159.5  4980.6  156.73  4986.2  148.47  5021.1  148.47
  5025.2  154.27    5035   159.3    5041  160.29  5084.1  158.95  5115.7  155.06
  5150.4   157.3  5158.8  155.29  5164.6  157.39  5180.3  154.68  5186.1  156.06
  5208.1   154.2  5223.4  154.55  5239.2  158.57  5509.1   159.8  5619.8  160.01
  5678.7  162.56  5782.3  161.47  5845.3  164.09  6000.4  167.62  6131.8  173.43
#Mann= 8 ,-1 , 0
    4546     .17       0  4744.7     .15       0  4894.3     .17       0
  4913.2     .15       0  4957.6     .09       0    5041     .15       0
  5509.1     .17       0  5782.3     .11       0
Bank Sta=4957.6,5041
XS Rating Curve= 0 ,0
Exp/Cntr=0.3,0.1

Type RM Length L Ch R = 1 ,51500   ,627,627,627
BEGIN DESCRIPTION:
CRYSTAL CREEK 102.0
END DESCRIPTION:
XS GIS Cut Line= 3
      3868528.55     10110176.05       3868218.3     10109561.75
      3867165.71     10109377.43
#Sta/Elev= 30
  4311.8  175.26  4435.2  175.65  4543.9  172.75  4768.6  164.59  4875.5  166.22
  4897.8  165.14    4920  157.69  4964.6  157.14  4970.2  154.14  4975.1  149.07
    5010  149.07  5020.8  156.31 5024.99157.1481  5061.4  158.71  5071.5  158.51
  5088.8  155.74  5093.9  156.92  5112.1  155.44  5153.4  158.35  5267.2  156.91
  5294.9  158.94  5335.5  157.38  5362.6  158.04  5494.8  160.08  5508.1  158.91
  5690.8  159.46  5744.1  161.49  5760.6  161.38  6025.8  172.23  6068.6  172.71
#Mann= 8 ,-1 , 0
  4311.8     .17       0  4543.9     .15       0  4768.6     .17       0
  4964.6     .09       0 5024.99     .15       0  5362.6     .11       0
  5744.1     .17       0  5760.6     .11       0
Bank Sta=4964.6,5024.99
XS Rating Curve= 0 ,0
Exp/Cntr=0.3,0.1

Type RM Length L Ch R = 1 ,50873   ,356,356,356
BEGIN DESCRIPTION:
CRYSTAL CREEK 101.0
END DESCRIPTION:
XS GIS Cut Line= 3
      3868964.27     10109664.98      3868057.37     10109187.32
      3867117.94     10109199.47
#Sta/Elev= 30
    3975  178.55  4029.9  177.56    4113  176.34  4293.8  173.35  4456.9  168.25
  4508.5  165.31  4552.5  156.89  4574.6  157.31    4590  159.17  4649.1  158.15
  4833.3  159.59  4841.2  158.33  4886.4   159.1  4899.4  157.86  4954.2  157.85
  4981.9  153.71  4991.7  147.34  5027.3  147.34  5028.3  147.84  5029.5   152.4
  5049.5  157.49  5098.3  158.33  5119.5  158.45  5129.5  157.34  5184.5  158.13
  5339.5  157.77  5458.9  161.97  5579.3  165.62  5680.6  166.07  5939.5   173.9
#Mann= 10 ,-1 , 0
    3975     .17       0  4029.9     .11       0    4113     .17       0
    4590     .15       0  4954.2     .09       0  5049.5     .15       0
  5098.3     .17       0  5184.5     .11       0  5458.9     .17       0
  5579.3     .11       0
Bank Sta=4954.2,5049.5
XS Rating Curve= 0 ,0
Exp/Cntr=0.3,0.1

Type RM Length L Ch R = 1 ,50517   ,517,517,517
BEGIN DESCRIPTION:
CRYSTAL CREEK 100.0
END DESCRIPTION:
XS GIS Cut Line= 3
      3869018.99     10109177.77      3868260.33     10108938.49
      3867153.74       10109055.
#Sta/Elev= 30
  4204.5  176.13  4216.2  173.28    4270   173.7  4347.1  172.67  4372.3  173.58
  4436.4   171.7  4512.2  167.89  4625.1  159.08    4690  157.33  4809.6  158.47
  4831.8  155.34  4846.2  153.89  4873.3  159.87  4897.7  156.49  4910.9   158.8
  4950.2  158.13  4960.7  156.17  4974.3   147.1  5009.9   147.1  5012.5  151.27
  5022.6  153.89  5075.2  156.63  5163.1  155.77    5261  158.76  5314.2   161.8
  5381.5  161.46  5487.6  161.54  5809.1  165.12  5977.9  167.48  6112.7  171.89
#Mann= 12 ,-1 , 0
  4204.5     .17       0    4270     .11       0  4347.1     .17       0
    4690     .15       0  4809.6     .11       0  4831.8     .15       0
  4960.7     .09       0  5075.2     .15       0    5261     .17       0
  5381.5     .11       0  5487.6     .17       0  5809.1     .11       0
Bank Sta=4960.7,5075.2
XS Rating Curve= 0 ,0
Exp/Cntr=0.3,0.1

Type RM Length L Ch R = 1 ,50000   ,555,555,555
BEGIN DESCRIPTION:
CRYSTAL CREEK 99.0
END DESCRIPTION:
XS GIS Cut Line= 3
      3869244.69     10109099.65      3868148.19     10108483.61
      3867187.35     10108687.33
#Sta/Elev= 30
  3742.3  174.41  3962.7  163.16    4039  160.56  4151.6  161.36  4195.2   159.5
    4201  157.51  4216.9  160.29    4327  157.28  4406.3  155.24  4518.5  158.12
  4627.5  156.06  4670.9  158.36  4782.5  155.52  4827.1  158.08  4920.1   157.7
    4966  154.85  4973.1  154.24  4979.7  145.94  5015.3  145.94  5020.8  151.29
    5031  155.44  5058.3  163.31  5116.1  164.53  5256.1  165.14  5452.9  166.12
  5511.5     169  5613.7   169.3  5746.6  165.61  5916.9  169.58  5982.2  170.31
#Mann= 10 ,-1 , 0
  3742.3     .17       0  3962.7     .11       0    4327     .17       0
  4518.5     .15       0    4966     .09       0    5031     .15       0
  5116.1     .17       0  5256.1     .11       0  5452.9     .17       0
  5916.9     .11       0
Bank Sta=4966,5031
XS Rating Curve= 0 ,0
Exp/Cntr=0.3,0.1

Type RM Length L Ch R = 1 ,49445   ,445,445,445
BEGIN DESCRIPTION:
CRYSTAL CREEK 98.0
END DESCRIPTION:
XS GIS Cut Line= 3
       3869587.6     10108813.21      3868321.65     10108118.38
      3867063.85     10108337.83
#Sta/Elev= 30
  3750.8  170.92  3907.8  162.91  4107.5   157.4  4304.9   158.9    4549  156.63
  4576.9  154.29  4598.7  157.08  4750.5  157.18  4870.6  155.07  4924.6  156.99
  4995.7  147.71  5017.5  152.98  5077.2   155.7  5093.3  152.38    5099  155.13
  5115.1  151.55  5119.1  147.04  5154.7  147.04  5155.7  147.54  5158.7  155.91
  5180.5  153.85  5219.1  157.27  5361.2  151.39  5391.6  157.29  5422.1  161.53
  5611.9  163.77  5746.9  166.89  5914.3  166.29  6216.8  165.96  6471.7  170.31
#Mann= 8 ,-1 , 0
  3750.8     .11       0  4107.5     .17       0  4750.5     .15       0
  4924.6     .09       0  5391.6     .17       0  5611.9     .11       0
  5914.3     .17       0  6216.8     .11       0
Bank Sta=4924.6,5391.6
XS Rating Curve= 0 ,0
Exp/Cntr=0.3,0.1

Type RM Length L Ch R = 1 ,49000   ,500,500,500
BEGIN DESCRIPTION:
CRYSTAL CREEK 97.0
END DESCRIPTION:
XS GIS Cut Line= 3
      3869517.82     10107911.07      3868718.51      10107839.6
      3867008.44     10108059.86
#Sta/Elev= 30
  4197.5  176.94  4258.2  177.29  4428.4  172.22  4548.9  166.08  4587.2  161.99
  4639.2  161.28  4719.5  153.85  4812.8  153.88  4950.5  156.62  4960.5  155.07
  4970.5  149.91  4971.8  145.58  4972.8  145.08  5008.4  145.08  5010.7  148.54
  5020.8  153.59  5030.9  154.71  5172.1  155.05  5202.3  157.94  5242.6  158.69
  5454.9  156.86  5555.2  157.72  5704.9  162.62    5833  164.29  5857.7  162.65
    6019  167.37  6129.9  165.23  6321.5  166.28  6458.6  164.37  6724.2  169.46
#Mann= 6 ,-1 , 0
  4197.5     .17       0  4812.8     .15       0  4960.5     .09       0
  5030.9     .15       0  5454.9     .17       0  5704.9     .11       0
Bank Sta=4960.5,5030.9
XS Rating Curve= 0 ,0
Exp/Cntr=0.3,0.1

Type RM Length L Ch R = 1 ,48500   ,500,500,500
BEGIN DESCRIPTION:
CRYSTAL CREEK 96.0
END DESCRIPTION:
XS GIS Cut Line= 3
      3869493.52     10107364.47      3868726.39     10107426.07
       3867051.7     10107871.84
#Sta/Elev= 30
  4230.4   175.5  4326.4  174.52  4373.4  169.35  4587.2  153.81    4716  152.09
  4868.1  153.44  4898.2  148.59  4908.2  148.56  4928.3  149.14  4948.4  152.93
  4968.4   152.6  4978.5  148.36  4982.1   144.7  5017.8   144.7  5018.8   145.2
  5019.2  149.51  5029.5  153.42  5060.6  156.02  5076.9  154.84  5174.4  156.62
  5197.3  159.71  5264.4  158.87  5307.4  157.41  5484.9  159.53  5598.7  157.69
  5705.2  161.13  6033.3  166.47  6602.5  164.68  6612.8  166.73    6733  168.68
#Mann= 6 ,-1 , 0
  4230.4     .17       0    4716     .15       0  4968.4     .09       0
  5029.5     .15       0  5264.4     .17       0  5705.2     .11       0
Bank Sta=4968.4,5029.5
XS Rating Curve= 0 ,0
Exp/Cntr=0.3,0.1

Type RM Length L Ch R = 1 ,48000   ,782,782,782
BEGIN DESCRIPTION:
CRYSTAL CREEK 95.0
END DESCRIPTION:
XS GIS Cut Line= 3
      3869319.94     10106661.33      3868600.76     10107079.85
      3867048.49     10107805.48
#Sta/Elev= 30
  4167.9   168.9  4254.9  164.89  4309.2  165.07  4331.5  161.03  4454.2  156.79
  4482.7  156.69    4492  154.87  4497.8  151.25  4540.8  156.44  4689.7  155.98
  4754.3     152  4828.7  154.95  4967.7  153.56  4973.5  152.26  4980.9  143.88
  5016.7  143.88  5025.3  148.77  5057.4  150.19  5080.2  153.63  5134.8  153.19
  5200.8  153.37  5290.2   159.9  5536.4  160.94  5665.5  158.95  5890.1   166.5
  5949.7  166.73  5955.6  166.76  6095.7  164.75  6551.9  164.25  6713.5  168.39
#Mann= 9 ,-1 , 0
  4167.9     .11       0  4254.9     .17       0  4454.2     .15       0
  4967.7     .09       0  5080.2     .15       0  5134.8     .17       0
  5200.8     .11       0  5949.7     .17       0  5955.6     .11       0
Bank Sta=4967.7,5080.2
XS Rating Curve= 0 ,0
Exp/Cntr=0.3,0.1

Type RM Length L Ch R = 1 ,47218   ,548,548,548
BEGIN DESCRIPTION:
CRYSTAL CREEK 94.0
END DESCRIPTION:
XS GIS Cut Line= 3
      3868859.86     10106249.01      3868482.92     10106451.96
      3867375.95     10107471.73
#Sta/Elev= 30
  4571.9  174.47    4572  174.47  4780.5  174.69  4862.4   166.6  4878.6  164.39
  4888.7  160.43  4928.1  151.57  4960.3  151.41  4971.9  147.99  4976.4  142.73
  5012.3  142.73  5017.3  149.31  5038.2  152.74  5088.2  150.23  5130.1  152.53
  5215.2  149.71  5286.1  154.37  5330.7  154.09  5466.4  154.44  5625.7  153.78
  5675.1  155.41  5731.8  153.92  5946.4  153.67    5991  153.82  6050.5  152.79
  6085.8  154.57  6199.1  163.14    6269  164.52  6425.3  163.14  6505.1  165.62
#Mann= 11 ,-1 , 0
  4571.9     .11       0    4572     .17       0  4888.7     .15       0
  4960.3     .09       0  5038.2     .15       0  5330.7     .17       0
  5466.4     .11       0  5946.4     .17       0    5991     .11       0
  6085.8     .17       0    6269     .11       0
Bank Sta=4960.3,5038.2
XS Rating Curve= 0 ,0
Exp/Cntr=0.3,0.1

Type RM Length L Ch R = 1 ,46670   ,139,139,139
BEGIN DESCRIPTION:
CRYSTAL CREEK 93.0
END DESCRIPTION:
XS GIS Cut Line= 3
      3868644.16     10105847.53      3868134.51     10106143.19
      3867195.65     10107290.13
#Sta/Elev= 30
  4410.8  168.59  4521.9  160.99  4725.6  154.32    4849  159.04  4886.2  157.14
    4902  152.86    4945  151.05  4977.2  142.95  5013.2  142.95  5017.5  149.38
    5024  151.15  5081.4  149.07  5209.2   153.4  5223.5  150.03  5273.1  152.47
  5280.9  150.52  5287.4  152.66  5316.1  149.91  5351.3  154.64    5380  150.05
  5450.3  149.55    5586  152.96  5656.3  151.52  5685.1  155.31  5734.6   151.1
  5940.6  154.14  5954.9  152.16  6055.4  157.91  6325.3  160.15  6482.2  164.78
#Mann= 3 , 0 , 0
  4410.8     .11       0    4945     .09       0    5024     .11       0
Bank Sta=4945,5024
XS Rating Curve= 0 ,0
Exp/Cntr=0.3,0.1

Type RM Length L Ch R = 1 ,46531   ,531,531,531
BEGIN DESCRIPTION:
CRYSTAL CREEK 92.0
END DESCRIPTION:
XS GIS Cut Line= 3
       3868474.3     10105688.15      3867992.67     10106090.52
      3866995.46     10107196.15
#Sta/Elev= 30
  4372.4  167.35  4521.4  157.68  4698.4  155.54  4733.5  157.46  4762.2  154.36
  4833.7  154.58  4961.3  148.73  4975.6  147.03  4978.4  142.81  5014.4  142.81
  5015.4  143.31  5017.8  148.57  5025.3  149.13  5081.5  148.73  5088.8  150.11
  5095.5  148.96  5131.4  151.91  5194.9  149.09  5244.2  151.88  5336.9  149.91
  5378.8  151.01  5485.5  148.17  5532.9  150.91  5591.7   154.7  5612.7  152.46
  5803.6  151.97  5938.5  154.53  6030.4   154.1  6264.4  162.19  6488.9  165.17
#Mann= 5 ,-1 , 0
  4372.4     .11       0  4961.3     .09       0  5025.3     .11       0
  5532.9     .17       0  5803.6     .11       0
Bank Sta=4961.3,5025.3
XS Rating Curve= 0 ,0
Exp/Cntr=0.3,0.1

Type RM Length L Ch R = 1 ,46000   ,500,500,500
BEGIN DESCRIPTION:
CRYSTAL CREEK 91.0
END DESCRIPTION:
XS GIS Cut Line= 3
      3868034.75     10105584.53      3867609.49     10105958.34
      3866855.26     10106807.29
#Sta/Elev= 30
  4433.8  167.74  4620.3  158.97  4698.1  161.78  4719.9  157.15  4762.5  159.36
  4798.5  156.81  4826.2  151.64  4840.4  151.39  4868.9  143.48  4889.8   143.5
  4910.7  151.08  4960.9  150.41  4980.3  142.34  5016.3  142.34  5024.4  149.48
  5031.1  150.59  5060.2  147.32  5151.5  151.92  5286.1  149.99  5328.8   152.4
  5385.6  151.94  5442.5  147.07  5512.7  146.34  5569.6  152.16  5622.5  149.56
  5652.6  150.78  5810.5   151.7  5917.9  157.61  6092.2  164.55  6135.6  165.99
#Mann= 9 ,-1 , 0
  4433.8     .11       0  4798.5     .15       0  4960.9     .09       0
  5031.1     .15       0  5060.2     .11       0  5622.5     .17       0
  5652.6     .11       0  5917.9     .17       0  6092.2     .11       0
Bank Sta=4960.9,5031.1
XS Rating Curve= 0 ,0
Exp/Cntr=0.3,0.1

Type RM Length L Ch R = 1 ,45500   ,1000,1000,1000
BEGIN DESCRIPTION:
CRYSTAL CREEK 90.0
END DESCRIPTION:
XS GIS Cut Line= 3
      3868021.76     10105493.38      3867372.86     10105581.08
       3866624.2     10106396.12
#Sta/Elev= 30
  4345.2  166.55  4453.9  161.05  4601.4  156.66  4621.6  154.42  4641.8  149.55
  4665.5  148.17  4712.4  150.74  4762.9   150.3  4793.1  153.13  4815.8  151.25
  4904.1  150.28  4961.1  142.79  4966.9  139.64  5002.9  139.64  5031.8  150.71
  5058.2  149.59  5123.6  147.98  5137.8  149.28  5272.2  150.91  5350.5  148.94
  5420.9  151.59  5486.1  149.87  5555.8  146.74  5597.8  150.99  5711.2  156.94
  5739.6  159.99  5824.7  161.75  5902.3  166.23  6060.3  171.07  6106.7  172.86
#Mann= 7 ,-1 , 0
  4345.2     .11       0  4453.9     .17       0  4904.1     .09       0
  5031.8     .17       0  5058.2     .15       0  5486.1     .11       0
  6060.3    .125       0
Bank Sta=4904.1,5031.8
XS Rating Curve= 0 ,0
Exp/Cntr=0.3,0.1

Type RM Length L Ch R = 1 ,44500   ,500,500,500
BEGIN DESCRIPTION:
CRYSTAL CREEK 89.0
END DESCRIPTION:
XS GIS Cut Line= 3
      3868105.48     10105269.44      3866958.35     10105527.05
      3866312.27     10105979.06
#Sta/Elev= 30
  3824.3  164.06  4110.7  158.23  4242.1  156.97  4266.5  155.41  4309.8   148.4
  4324.1  149.49  4385.6  147.43  4457.3  150.24    4652   150.6  4676.9  149.96
    4693  147.33  4720.2  150.54  4805.8  151.78    4901  149.56  4959.5  148.92
  4969.8  146.93  4977.4  139.09  5013.5  139.09  5017.3  143.52    5025  147.31
  5061.6  148.89    5074  147.18  5124.6  148.53  5172.1  147.35  5183.7  145.93
  5219.6  154.89  5232.5  156.27    5332  158.74  5535.3  158.63  5788.5  169.15
#Mann= 7 ,-1 , 0
  3824.3     .11       0  4110.7     .17       0    4901     .15       0
  4959.5     .09       0  5061.6     .15       0  5172.1     .11       0
    5332     .17       0
Bank Sta=4959.5,5061.6
XS Rating Curve= 0 ,0
Exp/Cntr=0.3,0.1

Type RM Length L Ch R = 1 ,44000   ,441,441,441
BEGIN DESCRIPTION:
CRYSTAL CREEK 88.0
END DESCRIPTION:
XS GIS Cut Line= 3
      3868109.38     10105214.73      3866787.54     10105227.23
      3866252.33     10105391.65
#Sta/Elev= 30
  3678.1  162.96  3759.6  159.43  3909.6     157  4013.6  158.62  4109.7  155.77
  4239.7  148.86  4279.7  148.59  4299.7  143.84  4319.7  149.55  4369.7  150.93
  4429.7  149.65  4509.7  151.22  4589.7  149.06  4709.7  150.23  4749.7   146.1
  4793.3  147.53  4909.7  147.98  4929.7  145.47  4969.7  146.83  4989.7  142.28
    4992  138.29  5028.2  138.29  5033.2  141.78  5041.5  143.95  5065.9  147.12
  5153.9  149.75  5208.9  159.79  5267.5   164.6  5365.6  169.04  5559.9  170.26
#Mann= 6 ,-1 , 0
  3678.1     .11       0  4013.6     .17       0  4793.3     .15       0
  4969.7     .09       0  5065.9     .15       0  5153.9     .11       0
Bank Sta=4969.7,5065.9
XS Rating Curve= 0 ,0
Exp/Cntr=0.3,0.1

Type RM Length L Ch R = 1 ,43559   ,559,559,559
BEGIN DESCRIPTION:
CRYSTAL CREEK 87.0
END DESCRIPTION:
XS GIS Cut Line= 3
      3868112.87     10105009.87      3866990.48      10104887.9
      3866367.81     10104911.07
#Sta/Elev= 30
    3871  162.24  3976.6   157.7  4057.1  158.62  4308.6  153.18  4439.3  147.25
  4459.6  148.82  4554.6  149.33  4600.3  144.03  4646.1  148.81  4670.7  149.16
  4751.2  146.18  4845.5  146.43  4881.9  146.03    4892  144.59  4942.3  144.27
  4972.5  142.51  5004.5  138.01  5040.7  138.01  5041.7  138.51  5042.7  146.24
  5052.7  146.78  5138.4  150.16  5157.7  151.08  5223.8  154.72  5262.8  159.26
  5282.8  158.36  5312.8   161.4  5336.2  160.64    5523  167.15  5623.1   168.1
#Mann= 8 ,-1 , 0
    3871     .11       0  4459.6     .17       0  4845.5     .15       0
  4881.9     .09       0  5052.7     .15       0  5138.4     .17       0
  5157.7     .15       0  5336.2     .17       0
Bank Sta=4881.9,5052.7
XS Rating Curve= 0 ,0
Exp/Cntr=0.3,0.1

Type RM Length L Ch R = 1 ,43000   ,500,500,500
BEGIN DESCRIPTION:
CRYSTAL CREEK 86.0
END DESCRIPTION:
XS GIS Cut Line= 3
      3868162.91      10104766.9      3867126.26     10104614.48
      3866417.86     10104511.07
#Sta/Elev= 30
  3952.2  165.75  4174.1  157.78  4290.9  157.01    4503  148.21  4654.7  148.05
  4685.1  145.77  4839.6  143.44  4846.6  142.63  4856.9  145.75  4947.8  146.77
    4958  146.67    4968  137.49  5004.2  137.49  5028.7  145.48  5038.8  146.42
  5048.9  145.49  5056.1  141.78  5061.1  144.58  5079.2  143.87  5109.6     147
  5126.1  144.55  5160.1  148.45  5180.3  148.23  5196.1  144.61  5201.1  149.38
    5251  146.79    5261  149.15  5264.9  147.41    5336   155.3  5715.9  166.44
#Mann= 6 ,-1 , 0
  3952.2     .11       0  4174.1     .17       0  4839.6     .15       0
  4947.8     .09       0  5038.8     .15       0  5264.9     .17       0
Bank Sta=4947.8,5038.8
XS Rating Curve= 0 ,0
Exp/Cntr=0.3,0.1

Type RM Length L Ch R = 1 ,42500   ,500,500,500
BEGIN DESCRIPTION:
CRYSTAL CREEK 85.0
END DESCRIPTION:
XS GIS Cut Line= 3
      3868067.87     10104261.07      3867261.18      10104204.1
      3866417.81     10104411.08
#Sta/Elev= 30
  4191.3  171.01  4251.5  169.08  4331.7  162.99    4472  155.46  4762.7  151.27
  4868.6  146.84  4913.1  144.98  4953.2     146  4963.2  143.41  4964.1  136.73
  4965.1  136.23  5001.4  136.23  5004.1  139.21  5008.4  138.27  5034.3  144.57
  5065.2   144.1  5085.8  139.18  5091.6  142.51  5096.7  139.79  5106.4  141.63
    5127  142.74  5138.3  145.85  5165.5  146.15  5465.7  156.79  5470.9  155.77
  5548.8  156.71    5554  155.07  5559.5  155.23  5595.6   157.7  5868.4   166.7
#Mann= 5 ,-1 , 0
  4191.3     .17       0  4868.6     .15       0  4953.2     .09       0
  5034.3     .15       0  5165.5     .17       0
Bank Sta=4953.2,5034.3
XS Rating Curve= 0 ,0
Exp/Cntr=0.3,0.1

Type RM Length L Ch R = 1 ,42000   ,442,442,442
BEGIN DESCRIPTION:
CRYSTAL CREEK 84.0
END DESCRIPTION:
XS GIS Cut Line= 3
      3868089.42      10104129.2      3867354.39     10103830.53
      3866448.06     10104016.44
#Sta/Elev= 30
  4206.6  171.03  4251.5   170.2  4321.4   165.3  4350.9  165.52    4381  160.03
  4493.7  151.89  4559.7  149.72  4637.3  151.26  4675.3   149.6  4910.4  152.33
  4953.1  147.32    4964   143.8  4974.7  142.08  4976.3  136.27  4977.3  135.77
  5013.6  135.77  5014.6  136.27  5016.9     142  5024.8  144.58  5047.5  145.35
  5098.5   141.8  5149.6   146.4  5181.1  140.07  5205.8  147.01  5282.3  146.91
  5312.9  143.68  5333.3  146.03  5579.2  156.46  5751.9  156.77  5925.2  162.04
#Mann= 6 ,-1 , 0
  4206.6     .17       0  4493.7     .15       0  4675.3     .17       0
    4964     .09       0  5024.8     .17       0  5205.8     .17       0
Bank Sta=4964,5024.8
XS Rating Curve= 0 ,0
Exp/Cntr=0.3,0.1

Type RM Length L Ch R = 1 ,41558   ,890,890,890
BEGIN DESCRIPTION:
CRYSTAL CREEK 83.0
END DESCRIPTION:
XS GIS Cut Line= 3
      3868713.56     10103537.65      3867304.29     10103432.36
      3866417.87     10103761.06
#Sta/Elev= 30
  3586.8  162.63  3745.1  153.74  3883.3  150.23  4063.8  151.17  4164.1  149.47
  4424.8  153.42  4655.5  151.78  4866.1  152.76  4896.1  151.26  4926.2  144.51
  4956.3  143.41  4976.4  138.03  4976.6   135.9  4977.6   135.4  5013.9   135.4
  5014.9   135.9  5017.5  143.89  5036.5  143.37  5072.2  145.92  5152.7  143.15
    5183  145.41  5316.2  145.64  5390.8   142.9  5414.1  145.22  5531.6  148.08
  5642.4  155.06  5703.2  156.78  5721.4  159.04  5897.4  164.39  5945.4  165.42
#Mann= 5 ,-1 , 0
  3586.8     .17       0  4956.3     .09       0  5017.5     .17       0
  5414.1     .17       0  5897.4     .11       0
Bank Sta=4956.3,5017.5
XS Rating Curve= 0 ,0
Exp/Cntr=0.3,0.1

Type RM Length L Ch R = 1 ,40668   ,168,168,168
BEGIN DESCRIPTION:
CRYSTAL CREEK 82.0
END DESCRIPTION:
XS GIS Cut Line= 3
      3868648.98     10102948.32      3867223.98     10102889.71
       3866241.5     10102883.22
#Sta/Elev= 30
  3573.8  160.13  3755.1  151.24  4112.8  149.22  4135.4  146.97  4245.5   151.8
  4375.6  146.25  4405.6  150.16  4455.7  150.56  4539.7  146.93  4625.8   141.9
    4796  143.94  4843.1  141.38  4956.1  144.58  4987.9  134.68  5024.3  134.68
  5025.3  135.18  5026.1  142.56  5036.1  143.03  5066.1  139.51  5275.6  143.11
  5394.4  150.65    5493  153.93  5591.6   155.5  5636.1  155.97  5646.1  153.08
  5666.1   157.7  5736.1  160.54  5749.1  158.71  5926.2  166.52  5982.5  165.99
#Mann= 9 ,-1 , 0
  3573.8     .17       0  4539.7     .15       0  4956.1     .09       0
  5036.1     .15       0  5275.6     .17       0  5394.4     .11       0
    5493     .17       0  5591.6     .11       0  5749.1     .17       0
Bank Sta=4956.1,5036.1
XS Rating Curve= 0 ,0
Exp/Cntr=0.3,0.1

Type RM Length L Ch R = 1 ,40500   ,387,387,387
BEGIN DESCRIPTION:
CRYSTAL CREEK 81.0
END DESCRIPTION:
XS GIS Cut Line= 3
      3868619.73     10102753.53      3867178.33     10102736.52
      3866221.65     10102711.89
#Sta/Elev= 30
  3558.5  167.79  3700.4  161.72  3950.4  158.47  4000.4  155.89  4060.4  155.83
  4160.4  150.73    4193  151.17  4240.4  149.14  4273.5  149.99  4350.4  143.14
  4650.5  143.21  4710.5  140.63  4760.5  143.84  4900.5  144.88  4950.5  143.52
  4970.5  141.13  4979.5  133.87  5015.9  133.87  5021.5  140.21  5030.5  142.99
  5040.5  143.65  5060.5  141.47  5070.5  143.58  5130.5  146.66  5244.2  149.97
  5583.3  155.59  5630.7  156.21  5880.8   167.3  5930.8  166.42    5957  167.56
#Mann= 6 ,-1 , 0
  3558.5     .17       0  4273.5     .15       0  4950.5     .09       0
  5040.5     .15       0  5244.2     .17       0  5583.3     .11       0
Bank Sta=4950.5,5040.5
XS Rating Curve= 0 ,0
Exp/Cntr=0.3,0.1

Type RM Length L Ch R = 1 ,40113   ,613,613,613
BEGIN DESCRIPTION:
CRYSTAL CREEK 80.0
END DESCRIPTION:
XS GIS Cut Line= 3
      3868341.94     10102392.42      3867028.04     10102394.49
      3866328.09     10102416.72
#Sta/Elev= 30
  3686.1  168.23  3750.2  167.48  3960.2  153.14  4040.2  151.03  4350.2  148.49
    4581  150.24  4660.2   148.2  4710.2  151.48  4740.2  151.55  4780.2  146.67
  4820.2  139.17  4840.2  138.05  4860.2  141.91  4880.2  139.65  4900.2  142.99
  4970.2  142.03  4979.3  132.94  5015.9  132.94  5020.2  139.66 5026.41 141.877
  5040.2  144.22  5081.2  143.86  5150.3  148.04  5280.3  151.13  5290.3  150.71
  5310.3  145.49  5330.4  147.05  5365.1  152.95  5575.3   160.7  5700.3  166.24
#Mann= 6 ,-1 , 0
  3686.1     .17       0    4581     .15       0  4970.2     .09       0
 5026.41     .15       0  5081.2     .17       0  5575.3     .11       0
Bank Sta=4970.2,5026.41
XS Rating Curve= 0 ,0
Exp/Cntr=0.3,0.1

Type RM Length L Ch R = 1 ,39500   ,500,500,500
BEGIN DESCRIPTION:
CRYSTAL CREEK 79.0
END DESCRIPTION:
XS GIS Cut Line= 3
      3868167.84     10101961.07      3867238.34       10102072.
      3866367.88     10101961.07
#Sta/Elev= 30
  4063.9   161.8  4144.5  159.26  4195.2  155.72    4225  155.64  4265.3  152.13
  4277.6  149.75  4355.1  151.67  4396.2  148.52  4456.7  149.99  4597.7  146.63
  4782.6  146.76  4889.7  144.13  4940.1   145.3  4952.6  144.53  4957.3141.6546
  4970.3   136.6  4971.1  132.49  4972.1  131.99  5008.7  131.99  5009.7  132.49
  5010.6  137.81  5020.7   141.5  5161.8  144.25  5212.2  144.38  5302.9  141.81
  5366.4  143.94  5635.6  152.95  5786.8  160.22  5827.1  164.21  5877.5  164.83
#Mann= 4 ,-1 , 0
  4063.9     .17       0  4957.3     .09       0  5020.7     .15       0
  5366.4     .17       0
Bank Sta=4957.3,5020.7
XS Rating Curve= 0 ,0
Exp/Cntr=0.3,0.1

Type RM Length L Ch R = 1 ,39000   ,457,457,457
BEGIN DESCRIPTION:
CRYSTAL CREEK 78.0
END DESCRIPTION:
XS GIS Cut Line= 3
      3868167.85     10101811.07      3866995.84     10101734.73
      3866362.78     10101850.75
#Sta/Elev= 30
  3825.5  161.47  3855.6  163.09  3935.7  162.09  4156.2  149.23  4266.4  147.27
  4346.6  148.63  4416.8  147.93    4557   143.1  4630.9  143.97  4707.4  142.21
  4857.7  144.85  4867.7  142.26  4887.7  136.65  4907.8  133.79  4927.8  132.01
  4947.9  132.33  4949.6  131.02  4986.3  131.02    4988  132.99    5000  132.27
  5018.3  133.63  5048.8  140.11  5063.5  141.63  5089.4  135.39  5098.7     135
  5121.7  136.09  5140.3  140.81  5180.9  145.19  5323.3  149.33  5643.6  163.86
#Mann= 5 ,-1 , 0
  3825.5     .17       0  4630.9     .15       0  4867.7     .09       0
  5063.5     .15       0  5098.7     .17       0
Bank Sta=4867.7,5063.5
XS Rating Curve= 0 ,0
Exp/Cntr=0.3,0.1

Type RM Length L Ch R = 1 ,38543   ,543,543,543
BEGIN DESCRIPTION:
CRYSTAL CREEK 77.0
END DESCRIPTION:
XS GIS Cut Line= 3
      3868140.55     10101691.02       3866813.9     10101362.16
      3866397.56     10101395.89
#Sta/Elev= 30
  3633.2  159.69  3646.3  161.98  3677.2  161.69    3694  159.13  3699.1  160.85
  3735.4  159.94  3934.8  151.25  4058.4  148.61  4195.8  147.72  4402.7  149.66
  4563.1  141.56  4674.1  145.06  4738.9  143.41  4816.6  138.57  4851.7  141.31
  4934.1  138.42  4975.3   140.3  4995.4  133.52  4997.7  130.56  5034.4  130.56
  5035.4  131.06  5036.2  135.17  5044.8  137.87  5049.8  134.61  5056.2  141.15
  5096.4  139.32  5156.6  148.24    5323  159.19  5377.3  163.16  5417.7  163.28
#Mann= 5 ,-1 , 0
  3633.2     .17       0  4674.1     .15       0  4975.3     .09       0
  5056.2     .15       0    5323     .11       0
Bank Sta=4975.3,5056.2
XS Rating Curve= 0 ,0
Exp/Cntr=0.3,0.1

Type RM Length L Ch R = 1 ,38000   ,500,500,500
BEGIN DESCRIPTION:
CRYSTAL CREEK 76.0
END DESCRIPTION:
XS GIS Cut Line= 3
      3868175.27     10101513.93      3866908.31     10100966.68
      3866543.36     10100993.11
#Sta/Elev= 30
  3619.9  159.97  3824.1  152.13  4039.8  149.07  4173.7  150.83  4249.6   146.6
  4412.3  146.82  4553.9  150.31    4741  149.08  4822.9  143.24  4837.1  138.76
  4851.8  140.76  4875.3  139.71  4880.8  136.87  4898.8  138.46  4904.3  136.64
  4913.4  140.38  4922.3  140.58  4935.1  138.06  4967.8  140.27  4989.6  137.27
  4991.1  131.19  4992.1  130.69  5028.8  130.69  5029.8  131.19  5030.5  135.11
  5050.6  141.18  5110.7  144.84    5201  154.09  5303.4   160.1  5365.9  161.85
#Mann= 5 ,-1 , 0
  3619.9     .17       0    4741     .15       0  4967.8     .09       0
  5050.6     .15       0  5303.4     .11       0
Bank Sta=4967.8,5050.6
XS Rating Curve= 0 ,0
Exp/Cntr=0.3,0.1

Type RM Length L Ch R = 1 ,37500   ,500,500,500
BEGIN DESCRIPTION:
CRYSTAL CREEK 75.0
END DESCRIPTION:
XS GIS Cut Line= 3
      3868258.71     10100628.29      3867037.23     10100551.42
      3866617.85     10100611.07
#Sta/Elev= 30
  3776.1  154.73  3997.4  150.54  4067.5   147.2  4087.6  148.37  4157.7   147.9
  4458.3  141.61  4588.6  143.41  4610.6  144.87  4698.8  144.53    4799  146.71
  4843.5  144.84  4925.1  140.46  4959.3  140.86  4979.3  137.97  5001.2  129.92
  5037.9  129.92  5038.9  130.42  5039.8  138.64  5089.2  136.93  5104.7  136.97
  5110.5  140.02  5120.6  141.32  5140.8  140.21  5201.4   144.2  5302.4   153.2
  5383.1  158.01  5388.2  155.48  5403.4  158.85  5421.3  159.84  5423.6  159.84
#Mann= 6 ,-1 , 0
  3776.1     .17       0  4843.5     .15       0  4979.3     .09       0
  5039.8     .15       0  5089.2     .17       0  5421.3     .11       0
Bank Sta=4979.3,5039.8
XS Rating Curve= 0 ,0
Exp/Cntr=0.3,0.1

Type RM Length L Ch R = 1 ,37000   ,500,500,500
BEGIN DESCRIPTION:
CRYSTAL CREEK 74.0
END DESCRIPTION:
XS GIS Cut Line= 3
      3868244.72     10100576.43      3867108.51      10100156.3
      3866687.55     10100189.93
#Sta/Elev= 30
  3788.6  155.96  3906.4  156.63  3974.6  154.19  4041.1  152.87  4158.4  147.18
  4211.7   148.6  4341.2  145.54  4488.9  147.15  4654.4  141.06  4734.2  141.21
  4819.5  145.32  4873.7  144.73  4917.4  144.12  4936.7  141.47  4942.5  138.76
  4958.1  136.51    4960  131.07    4961  130.57  4997.8  130.57    5000  133.37
  5040.8  138.68  5080.9  138.72  5131.1  143.19  5161.2  141.42  5181.2  144.07
  5209.5  139.73  5241.4  138.03  5374.8  149.15  5401.9     153  5422.3  153.41
#Mann= 7 ,-1 , 0
  3788.6     .11       0  3974.6     .17       0  4873.7     .15       0
  4942.5     .09       0  5040.8     .15       0  5209.5     .17       0
  5374.8     .11       0
Bank Sta=4942.5,5040.8
XS Rating Curve= 0 ,0
Exp/Cntr=0.3,0.1

Type RM Length L Ch R = 1 ,36500   ,512,512,512
BEGIN DESCRIPTION:
CRYSTAL CREEK 73.0
END DESCRIPTION:
XS GIS Cut Line= 3
      3868234.28     10099997.67      3867031.94     10099744.54
      3866677.01     10099942.08
#Sta/Elev= 30
  3771.3  154.89  3793.1  154.02  3931.2  149.38  3986.7  150.03  4136.7  147.21
  4258.2   144.1  4319.5  146.57  4463.5  145.68  4646.5  144.46  4741.2  147.19
  4769.1  149.28  4851.5  144.89  4871.3  139.51  4881.5  135.25    4902  133.42
    4946  133.99  4973.5  137.65  4983.7   136.6  4988.4  129.05  5025.2  129.05
  5038.8  135.51  5060.5   139.4  5066.2  137.48  5073.3  140.16  5109.7  138.83
    5178  140.95  5234.3  142.67  5266.3  147.86  5327.7  149.75  5406.2  152.96
#Mann= 10 ,-1 , 0
  3771.3     .11       0  3793.1     .17       0  3986.7     .11       0
  4136.7     .17       0  4463.5     .11       0  4741.2     .17       0
  4871.3     .09       0  5073.3     .15       0    5178     .17       0
  5327.7     .11       0
Bank Sta=4871.3,5073.3
XS Rating Curve= 0 ,0
Exp/Cntr=0.3,0.1

Type RM Length L Ch R = 1 ,35988   ,116,116,116
BEGIN DESCRIPTION:
CRYSTAL CREEK 72.0
END DESCRIPTION:
XS GIS Cut Line= 3
      3868289.56     10099180.03      3866968.87     10099281.75
      3866686.86     10099670.42
#Sta/Elev= 30
  3675.4  152.98  3727.3  149.23  3857.6  149.99  4008.1  143.17  4218.7  144.04
    4329  141.23  4449.4  145.32  4572.5  141.42    4650  135.81    4660  135.62
  4665.3  138.74  4670.3  136.12  4690.1  138.65  4750.3  132.83  4770.3  136.66
  4803.9  137.67  4840.5  136.43  4860.6  133.56  4900.7  139.31  4930.9  138.85
  4970.9  136.99  4979.6  130.21  5016.4  130.21  5028.7  136.04  5072.7  137.93
  5099.8  136.72  5164.7  141.37  5177.1  140.68  5200.3  142.96  5480.2  152.04
#Mann= 6 ,-1 , 0
  3675.4     .11       0  4572.5     .17       0  4803.9     .15       0
  4930.9     .09       0  5072.7     .15       0  5177.1     .17       0
Bank Sta=4930.9,5072.7
XS Rating Curve= 0 ,0
Exp/Cntr=0.3,0.1

Type RM Length L Ch R = 1 ,35872   ,233,233,233
BEGIN DESCRIPTION:
Mapping XS 6da51c09
END DESCRIPTION:
XS GIS Cut Line= 3
      3867973.38     10098291.43      3866968.01     10099165.64
      3866665.13     10099627.48
#Sta/Elev= 30
  3667.7  151.83  3749.4   146.3  3876.7  143.73  3940.3  145.65  4054.2  143.08
    4472  144.11  4606.9  139.17  4755.9  140.43  4868.9  138.45    4905  135.78
  4919.3  132.36  4940.1  136.27    4961   135.9  4968.6   131.2  4975.3  133.57
  4982.9  130.56  5022.6  127.87  5059.7  127.87  5060.7  128.37  5062.2  133.27
  5068.2  135.03  5119.5  137.46  5149.7  136.36  5176.7  142.42  5191.8   142.2
  5197.8  139.11  5221.8  145.31  5299.3  145.62  5357.2  148.54  5552.3  151.44
#Mann= 5 ,-1 , 0
  3667.7     .11       0    4961     .06       0  5068.2     .11       0
  5299.3     .17       0  5357.2     .11       0
Bank Sta=4961,5068.2
XS Rating Curve= 0 ,0
Exp/Cntr=0.3,0.1

Type RM Length L Ch R = 1 ,35639   ,253,253,253
BEGIN DESCRIPTION:
CRYSTAL CREEK 71.0
END DESCRIPTION:
XS GIS Cut Line= 3
      3867949.08     10098092.64       3866921.6     10098960.73
      3865714.81     10099870.17
#Sta/Elev= 30
  3654.9  152.92  3881.4  143.58  4389.1  140.98  4471.1  141.66  4522.5  142.35
  4655.9  137.36  4894.8  137.11  4932.1  137.79  4946.1  138.72  4981.3  133.03
  4991.4  127.23  5028.5  127.23  5030.7  133.88  5067.3  137.58  5117.4  135.12
  5213.5  140.34  5338.9  140.67  5474.2  147.49  5524.6  144.48  5588.8  140.57
  5694.9  134.85    5724  128.15  5738.6  136.66  5800.2   137.3  5943.8  138.72
  6102.9  146.69  6400.1  148.23  6438.1  149.13    6459  144.39  6511.1  153.41
#Mann= 15 ,-1 , 0
  3654.9     .11       0  4389.1     .17       0  4471.1     .11       0
  4522.5     .17       0  4655.9     .15       0  4894.8     .11       0
  4932.1     .15       0  4946.1     .09       0  5067.3     .15       0
  5213.5     .17       0  5524.6     .11       0  5588.8     .15       0
  5800.2     .11       0  5943.8     .17       0  6400.1     .11       0
Bank Sta=4946.1,5067.3
XS Rating Curve= 0 ,0
Exp/Cntr=0.3,0.1

Type RM Length L Ch R = 1 ,35386   ,361,361,361
BEGIN DESCRIPTION:
Mapping XS 0432b14f
END DESCRIPTION:
XS GIS Cut Line= 3
      3867700.05     10097768.82      3866723.74     10098819.29
      3865958.09     10099364.42
#Sta/Elev= 30
  3569.2  152.36  3777.3  141.16  3819.8  144.66  3912.2  141.45  4046.5  145.76
  4237.6  143.28  4320.6  146.13  4548.8  144.31  4577.2  140.25  4591.3  134.64
  4626.5     133  4739.9  132.42  4789.2  137.71  4923.8  136.17  4959.3  129.62
  4966.1  133.03  4975.8  126.37    5013  126.37  5015.8  133.41  5095.8  133.17
  5145.6   140.2  5198.2  138.89  5306.4     139  5538.4  138.15  5575.2  126.96
  5597.4  136.27  5765.3  140.38  5795.1  143.25  5926.3  152.85  5943.2  153.95
#Mann= 9 ,-1 , 0
  3569.2     .11       0  4320.6     .15       0  4577.2     .07       0
  5145.6     .15       0  5198.2     .17       0  5306.4     .15       0
  5765.3     .17       0  5795.1     .11       0  5926.3     .17       0
Bank Sta=4577.2,5145.6
XS Rating Curve= 0 ,0
Exp/Cntr=0.3,0.1

Type RM Length L Ch R = 1 ,35025   ,525,525,525
BEGIN DESCRIPTION:
CRYSTAL CREEK 70.0
END DESCRIPTION:
XS GIS Cut Line= 3
      3867659.47     10097692.45      3866406.18     10098774.86
      3865923.17     10098897.35
#Sta/Elev= 30
    3344  151.03  3528.8  141.26  3627.6  143.38  3670.3  140.89  3875.5  145.86
  4301.1  145.77  4343.9  143.54  4442.8  145.74  4747.3  145.61  4818.8  144.68
  4861.6  142.83  4925.2  134.83    4968  137.29  4982.3  135.24  4995.6  127.42
  5039.5   127.9  5045.2  128.44  5050.3  132.83  5086.1  132.59  5091.3   136.4
  5121.9  136.93  5142.7  133.52    5184  134.03  5190.4   125.9  5227.6   125.9
  5235.6  135.65  5244.9   136.8  5372.9  138.48  5413.9  146.52  5498.3  157.84
#Mann= 4 ,-1 , 0
    3344     .11       0  4747.3     .17       0  4818.8     .07       0
  5413.9     .11       0
Bank Sta=4818.8,5413.9
XS Rating Curve= 0 ,0
Exp/Cntr=0.3,0.1

Type RM Length L Ch R = 1 ,34500   ,500,500,500
BEGIN DESCRIPTION:
CRYSTAL CREEK 69.0
END DESCRIPTION:
XS GIS Cut Line= 3
      3867659.46     10097648.19      3866143.84      10098471.7
      3865891.92     10098435.57
#Sta/Elev= 30
  3275.1  150.76  3314.7  149.89  3374.5  144.93  3456.3  141.56  3549.7  141.27
  3587.4  142.71  3661.3   141.1  3925.7   144.7  4023.5     144  4051.1  140.29
  4096.3  143.67  4211.4  143.17  4405.5  141.05  4552.8   137.1    4785  136.23
  4847.5  134.92  4857.9  136.46    4893  135.07    4951   136.3  4961.3  135.24
  4971.8  126.52  5017.9  126.52  5026.3  135.39  5076.8  133.28  5127.3  136.25
  5137.4  138.63  5162.1  149.33    5198  153.95  5208.1  156.75  5254.5  151.09
#Mann= 8 ,-1 , 0
  3275.1     .11       0  3549.7     .17       0  3661.3     .11       0
  4211.4     .17       0    4785     .15       0    4951     .07       0
  5026.3     .15       0  5162.1     .11       0
Bank Sta=4951,5026.3
XS Rating Curve= 0 ,0
Exp/Cntr=0.3,0.1

Type RM Length L Ch R = 1 ,34000   ,500,500,500
BEGIN DESCRIPTION:
CRYSTAL CREEK 68.0
END DESCRIPTION:
XS GIS Cut Line= 3
      3867651.64     10097624.75      3866091.44     10098035.28
      3865602.28     10097936.17
#Sta/Elev= 30
  3386.7  150.51  3509.7  143.72  3624.4  141.95  3741.3  144.24  3782.6  143.39
  3902.6   142.7  3969.7   144.1  4023.6  142.93  4145.5  136.69  4345.7  136.57
  4448.8  135.42  4481.2  134.88  4653.4  136.18  4703.8  134.03  4723.7  131.08
  4789.2  135.21  4931.3  135.98    4952  132.96    4960  124.99  5006.1  124.99
  5013.9  129.45  5034.3  131.95    5048  135.96  5054.7  138.77  5093.6  141.77
  5264.7  144.06  5327.1  144.54  5364.6  144.71  5464.5  150.24  5499.1  152.83
#Mann= 13 ,-1 , 0
  3386.7     .11       0  3624.4     .17       0  3782.6     .11       0
  4345.7     .17       0  4448.8     .11       0  4481.2     .17       0
  4789.2     .15       0  4931.3     .07       0    5048     .15       0
  5264.7     .17       0  5327.1     .11       0  5364.6     .17       0
  5464.5     .11       0
Bank Sta=4931.3,5048
XS Rating Curve= 0 ,0
Exp/Cntr=0.3,0.1

Type RM Length L Ch R = 1 ,33500   ,500,500,500
BEGIN DESCRIPTION:
CRYSTAL CREEK 67.0
END DESCRIPTION:
XS GIS Cut Line= 3
      3867649.01     10097598.71      3866405.88     10097659.56
      3865584.75     10097896.32
#Sta/Elev= 30
  3768.2  150.46  3893.9  143.44  3949.6   142.9  3959.6  140.72  3992.9  142.55
  4049.7  143.98    4320  141.91    4340  143.73  4528.9  136.43  4685.6  141.39
  4784.5  138.48  4860.7  134.62  4910.7  135.59  4938.6  130.52  4943.7  132.78
  4986.3  124.04  5032.4  124.04    5042  127.92  5052.4  126.66  5070.2  132.79
  5075.4  129.94  5103.9  135.22  5114.8  132.97  5239.7  139.42  5406.2  141.47
  5645.2  140.73  5767.3  145.71  5811.4  148.83  5855.7  151.87  5867.4  152.85
#Mann= 10 ,-1 , 0
  3768.2     .11       0  3893.9     .17       0  3992.9     .11       0
  4685.6     .17       0  4784.5     .11       0  4910.7     .09       0
  5103.9     .15       0  5767.3     .17       0  5811.4     .11       0
  5855.7     .17       0
Bank Sta=4910.7,5103.9
XS Rating Curve= 0 ,0
Exp/Cntr=0.3,0.1

Type RM Length L Ch R = 1 ,33000   ,500,500,500
BEGIN DESCRIPTION:
CRYSTAL CREEK 66.0
END DESCRIPTION:
XS GIS Cut Line= 3
      3867302.65     10097049.35      3866358.15     10097240.29
      3865425.19     10097656.52
#Sta/Elev= 30
  4036.4  150.75  4225.9  142.44  4436.7  141.64  4497.7  141.47  4602.4  140.97
    4684   142.4  4806.5  141.34  4875.3  136.67  4888.1  132.88  4908.5  130.92
  4925.2  132.53  4969.7  133.44  4981.9  132.18  4990.1  127.12  4991.4  124.48
  4992.4  123.98  5038.6  123.98  5039.6  124.48  5044.2  134.96  5100.4  133.05
    5189   137.4  5229.9  137.96  5403.5  135.25    5515  135.14  5625.2  136.85
  5698.5  136.37  5756.7  137.96  5848.8  139.85  5900.7  146.41  6021.6  151.85
#Mann= 9 ,-1 , 0
  4036.4     .11       0  4436.7     .17       0  4497.7     .11       0
  4925.2     .15       0  4969.7     .09       0  5044.2     .15       0
  5100.4     .17       0  5625.2     .11       0  5756.7     .17       0
Bank Sta=4969.7,5044.2
XS Rating Curve= 0 ,0
Exp/Cntr=0.3,0.1

Type RM Length L Ch R = 1 ,32500   ,500,500,500
BEGIN DESCRIPTION:
CRYSTAL CREEK 65.0
END DESCRIPTION:
XS GIS Cut Line= 3
      3867288.76     10096924.35      3866164.91     10096855.04
      3865171.72     10097222.58
#Sta/Elev= 30
  3864.2   151.6  3999.6  148.73  4115.6  141.78  4238.1  141.11  4570.7  138.96
  4796.9  136.17  4823.9   133.4  4897.1  134.29  4927.1  130.83  4947.2  125.09
    4975   123.2  5021.2   123.2  5022.2   123.7  5023.2  129.82  5040.4  131.36
  5048.2  129.78  5072.4  134.31  5078.6   136.3    5109  136.45  5134.1   130.2
  5169.8  135.06  5210.9  133.75  5286.1  134.75  5397.1  132.22  5452.5  134.65
  5574.1  131.86    5660  133.31  5786.8  137.21  5881.9  145.44  6049.2  151.85
#Mann= 7 ,-1 , 0
  3864.2     .11       0  4238.1     .17       0  4570.7     .11       0
  4823.9     .15       0  4897.1     .09       0  5072.4     .15       0
  5210.9     .11       0
Bank Sta=4897.1,5072.4
XS Rating Curve= 0 ,0
Exp/Cntr=0.3,0.1

Type RM Length L Ch R = 1 ,32000   ,375,375,375
BEGIN DESCRIPTION:
CRYSTAL CREEK 64.0
END DESCRIPTION:
XS GIS Cut Line= 3
      3867333.83     10096788.92      3865987.19     10096430.21
        3865063.     10096955.62
#Sta/Elev= 30
  3606.4  150.56  3853.2   143.1  4008.5  143.88  4083.6  141.09    4304  140.14
  4331.2  141.01  4419.8  141.13  4549.5  134.04  4657.6  134.02  4678.5  131.11
  4699.2  133.67  4739.8  131.81  4795.4  134.01  4896.5  129.03  4940.4  127.82
  4975.3  130.04  4980.5  127.15    4989   127.4    4990  122.82    4991  122.32
  5037.3  122.32  5045.2  130.97  5127.3  133.15  5169.9  131.47  5213.1  139.25
    5278  144.13  5476.9  148.29  5675.9  148.42  5873.5  144.63  6063.1  149.03
#Mann= 9 ,-1 , 0
  3606.4     .11       0    4304     .17       0  4331.2     .11       0
  4657.6     .17       0  4795.4     .11       0  4896.5     .15       0
  4975.3     .09       0  5045.2     .15       0  5127.3     .11       0
Bank Sta=4975.3,5045.2
XS Rating Curve= 0 ,0
Exp/Cntr=0.3,0.1

Type RM Length L Ch R = 1 ,31625   ,136,136,136
BEGIN DESCRIPTION:
Mapping XS 75a4ff48
END DESCRIPTION:
XS GIS Cut Line= 4
      3867303.44     10096730.55      3865730.52     10096220.13
      3865435.38     10096126.38      3864827.76     10096692.34
#Sta/Elev= 30
  3322.8  148.45  3475.9  143.01  3756.5  144.61    3970  139.36  4049.5  141.49
  4169.7   137.8  4253.8  138.81  4278.5  138.19  4295.9  133.22  4316.9  138.88
  4494.2  141.75  4571.5   139.9  4630.2  134.56  4684.9  132.89  4947.7  132.23
  4960.4  130.65  4975.2  124.51  5001.5  123.04  5047.8  123.04  5048.8  123.54
  5051.7  131.87    5186   139.3    5211  139.98  5309.1  140.75    5486  137.32
  5570.5   139.8  5655.5  137.58  5818.2  138.24  6002.4  143.24  6116.5  149.39
#Mann= 5 ,-1 , 0
  3322.8     .11       0  4494.2     .17       0  4571.5     .09       0
    5186     .15       0    5211     .11       0
Bank Sta=4571.5,5186
XS Rating Curve= 0 ,0
Exp/Cntr=0.3,0.1

Type RM Length L Ch R = 1 ,31489   ,489,489,489
BEGIN DESCRIPTION:
CRYSTAL CREEK 63.0
END DESCRIPTION:
XS GIS Cut Line= 4
       3867552.7     10096666.42      3865709.69     10096077.77
      3865501.36     10096018.74      3864772.88     10096666.07
#Sta/Elev= 30
  3063.8  149.02    3327  147.04  3446.8  143.24  3572.8  142.91  3750.6  139.26
    4183  139.21  4285.1  139.02  4549.9  140.72    4592  139.85  4608.3  138.21
  4677.7137.6023  4832.5  131.79    4885  133.83  4972.7  132.58  4979.5  131.44
  4987.7  122.04    5034  122.04  5039.1  128.59  5044.3  128.18  5052.4  131.44
  5214.3  137.65  5289.8  138.24    5304  141.13  5318.3  141.34  5530.7  136.84
  5587.5  138.27  5672.8  136.71  5885.2  138.08  6048.3  142.78  6189.6  151.08
#Mann= 7 ,-1 , 0
  3063.8     .11       0    4183     .17       0  4285.1     .11       0
  4549.9     .17       0    4592     .11       0  4677.7     .09       0
  5214.3     .11       0
Bank Sta=4677.7,5214.3
XS Rating Curve= 0 ,0
Exp/Cntr=0.3,0.1

Type RM Length L Ch R = 1 ,31000   ,428,428,428
BEGIN DESCRIPTION:
CRYSTAL CREEK 62.0
END DESCRIPTION:
XS GIS Cut Line= 3
      3867594.24     10095466.02       3865838.5     10095638.57
      3864726.22      10096632.7
#Sta/Elev= 30
  3235.8  151.16  3448.4  139.85  3533.6   136.5  3653.4  137.25  4126.5  135.23
    4237  138.87  4508.3  140.65  4628.9   136.9  4839.9   138.2  4948.5  131.35
  4950.4  131.13    4970  126.15  4974.7  120.84    5021  120.84    5022  121.34
  5023.6  130.96  5030.3  129.11  5037.8  131.79  5129.8  134.78  5164.9  130.81
  5186.6  133.61  5271.9  133.11  5413.2  129.21  5483.7  139.59  5529.3  138.34
  5632.2  141.37  5845.4  136.58    6128  137.73  6326.9  140.89  6491.8  151.73
#Mann= 8 ,-1 , 0
  3235.8     .17       0  3448.4     .15       0  3653.4     .17       0
  4948.5     .15       0  4950.4     .09       0  5023.6     .15       0
  5271.9     .17       0  5529.3     .11       0
Bank Sta=4950.4,5023.6
XS Rating Curve= 0 ,0
Exp/Cntr=0.3,0.1

Type RM Length L Ch R = 1 ,30572   ,72,72,72
BEGIN DESCRIPTION:
Mapping XS d79a1941
END DESCRIPTION:
XS GIS Cut Line= 4
      3867654.09     10094577.79      3865752.27     10095240.88
      3864810.38     10096489.23      3864694.05     10096614.25
#Sta/Elev= 30
  2985.9   150.4  3047.5  146.19  3352.6  135.31  3496.2  135.79  4046.2  136.25
  4124.8  136.06  4291.8  136.98  4350.1  136.36  4549.3  138.22  4782.3  135.39
  4856.4  137.93    4912  134.05    4925  132.92  4962.3  129.35  4970.9  119.71
  5017.2  119.71  5025.3  129.53  5046.5  132.15  5135.4  131.56  5202.6  132.83
  5246.3   130.8  5331.7  137.63  5396.2  139.55  5808.3  137.97  5945.7  139.86
  6066.5  136.64  6224.7  139.88  6480.7  138.21    6595   142.1  6734.6  152.86
#Mann= 12 ,-1 , 0
  2985.9     .17       0  3047.5     .11       0  3496.2     .15       0
  4046.2     .11       0  4124.8     .17       0  4291.8     .11       0
  4350.1     .17       0    4912     .15       0    4925     .09       0
  5046.5     .15       0  5135.4     .17       0  5808.3     .11       0
Bank Sta=4925,5046.5
XS Rating Curve= 0 ,0
Exp/Cntr=0.3,0.1
