HEC-RAS study CRYSTAL CREEK.prj: CRYSTAL CREEK Base Level Engineering

--- CRYSTAL CREEK.g10 (geometry) --- (continued)

Type RM Length L Ch R = 1 ,27394   ,394,394,394
BEGIN DESCRIPTION:
CRYSTAL CREEK 55.0
END DESCRIPTION:
XS GIS Cut Line= 3
      3864281.77     10093677.84      3863312.53      10094739.3
      3862892.93     10095295.84
#Sta/Elev= 30
  3562.6  154.99  3658.6  149.73  3808.5  138.14  3886.2  134.24  3971.3  136.19
  3992.3  133.94  4269.2  134.94  4344.7  135.52  4487.8  128.76  4574.5   130.7
  4686.1  125.54  4707.1  130.25  4726.7  128.62  4742.9   130.6  4848.9   130.9
  4877.3   129.8  4898.3  126.08  4912.5  130.26  4948.2  129.24  4969.2  122.56
    4974   115.9  5021.1   115.9  5026.8  122.97  5053.9  128.72  5108.7     133
  5209.3  141.19  5348.1  142.46  5425.3  144.66  5480.1  145.68    5697  150.54
#Mann= 13 ,-1 , 0
  3562.6     .12       0  3658.6     .05       0  4269.2     .12       0
  4344.7     .05       0  4574.5     .12       0  4726.7      .1       0
  4948.2     .07       0  5053.9      .1       0  5108.7     .12       0
  5209.3     .05       0  5348.1     .12       0  5425.3     .05       0
  5480.1     .12       0
Bank Sta=4948.2,5053.9
XS Rating Curve= 0 ,0
Exp/Cntr=0.3,0.1

Type RM Length L Ch R = 1 ,27000   ,500,500,500
BEGIN DESCRIPTION:
CRYSTAL CREEK 54.0
END DESCRIPTION:
XS GIS Cut Line= 3
      3864111.64     10093570.19      3863262.98     10094353.05
      3862649.83     10094941.73
#Sta/Elev= 30
  3845.4  151.51  4018.5  140.56  4207.3     134  4210.8  134.01  4294.6  129.77
  4337.2  133.96  4382.7  133.82  4414.8  134.76  4514.1  132.09  4535.1  128.88
  4697.8  125.99  4754.5  131.42  4811.2  128.07  4828.5  130.67  4874.7  124.78
  4952.6  127.31  4959.8  124.49  4966.6  125.55  4988.1  116.57  4999.8   115.5
  5046.9   115.5  5047.9     116  5051.7  127.11    5073  129.78  5122.4  128.36
  5143.8  129.78  5172.1  136.45  5221.7  137.95  5532.8  140.85    5850  155.44
#Mann= 8 ,-1 , 0
  3845.4     .05       0  4207.3     .12       0  4210.8     .05       0
  4382.7     .12       0  4828.5      .1       0  4952.6     .07       0
  5051.7      .1       0  5221.7     .12       0
Bank Sta=4952.6,5051.7
XS Rating Curve= 0 ,0
Exp/Cntr=0.3,0.1

Type RM Length L Ch R = 1 ,26500   ,500,500,500
BEGIN DESCRIPTION:
CRYSTAL CREEK 53.0
END DESCRIPTION:
XS GIS Cut Line= 3
      3864017.93     10093455.59      3863138.99     10093898.21
      3862117.86     10094561.06
#Sta/Elev= 30
  4015.9  155.07  4169.9  151.21  4355.3  135.12  4482.3  127.18  4654.2  125.38
  4705.4  125.84  4766.1  130.47  4891.2  131.13  4924.9 128.487  4973.1   121.4
  4987.3  114.83  5034.4  114.83  5047.1  124.32  5068.2  128.64  5083.4  125.96
  5119.6  132.66  5162.7  134.08  5213.2  130.76  5237.8     133  5270.6  135.32
    5322  132.85  5377.4   134.8  5395.6  135.13  5478.9  137.85  5509.2   141.5
  5530.3  138.08  5704.8  136.89  5892.8  142.74  6173.6  158.17  6217.4  157.74
#Mann= 9 ,-1 , 0
  4015.9     .05       0  4355.3     .12       0  4891.2      .1       0
  4924.9     .07       0  5068.2      .1       0  5162.7     .12       0
  5237.8     .05       0  5377.4     .12       0  5395.6     .05       0
Bank Sta=4924.9,5068.2
XS Rating Curve= 0 ,0
Exp/Cntr=0.3,0.1

Type RM Length L Ch R = 1 ,26000   ,500,500,500
BEGIN DESCRIPTION:
CRYSTAL CREEK 52.0
END DESCRIPTION:
XS GIS Cut Line= 3
      3864017.84     10093361.07      3863062.37     10093443.31
      3861872.44     10094198.42
#Sta/Elev= 30
    4041  155.21  4216.3  149.71  4496.9  128.81    4583  122.84  4620.3   124.9
  4673.3  128.69  4713.5  121.28  4793.8  122.36  4894.1   127.8  4944.3  127.26
  4974.4  121.85  4975.2  114.21  4976.2  113.71  5023.4  113.71  5029.4  116.11
  5052.7  119.54  5059.9  124.04  5070.3 127.376  5081.1  130.68  5111.6  127.71
  5193.1  129.46    5248  132.63  5344.6  132.37  5739.6  137.84  5821.5  137.27
  5857.9  134.49  5985.4  135.27  6038.8  135.95  6210.4  141.05  6409.3  150.46
#Mann= 10 ,-1 , 0
    4041     .05       0  4496.9     .12       0  4620.3      .1       0
  4944.3     .07       0  5070.3      .1       0  5193.1     .05       0
  5344.6     .12       0  5985.4     .05       0  6038.8     .12       0
  6210.4     .05       0
Bank Sta=4944.3,5070.3
XS Rating Curve= 0 ,0
Exp/Cntr=0.3,0.1

Type RM Length L Ch R = 1 ,25500   ,476,476,476
BEGIN DESCRIPTION:
CRYSTAL CREEK 51.0
END DESCRIPTION:
XS GIS Cut Line= 3
      3864021.38     10093316.72      3863295.96     10093097.58
      3861741.49     10093562.83
#Sta/Elev= 30
  4242.2  154.78  4425.7  148.29  4488.9  147.55  4620.8   139.2  4705.5  132.31
  4747.3  125.53  4838.3  124.96  4914.4   128.7  4956.2  124.99 4957.05 123.508
  4963.9   112.8  5011.2   112.8  5026.9  123.26  5065.2  126.04    5092  123.07
  5131.4  127.48  5169.7  125.28  5235.9  129.19  5330.2  129.01  5459.6  128.33
  5563.8  131.54  5659.1  130.61  5772.1  134.34  5958.3  137.28  6094.4  132.98
  6188.7  134.65  6271.5  134.79  6397.1  140.57  6605.4  152.55  6622.6  154.06
#Mann= 13 ,-1 , 0
  4242.2     .05       0  4425.7     .12       0  4838.3      .1       0
  4956.2     .07       0  5026.9      .1       0  5330.2     .12       0
  5459.6     .05       0  5563.8     .12       0  5772.1     .05       0
  6094.4     .12       0  6188.7     .05       0  6397.1     .12       0
  6605.4     .05       0
Bank Sta=4957.05,5026.9
XS Rating Curve= 0 ,0
Exp/Cntr=0.3,0.1

Type RM Length L Ch R = 1 ,25024   ,509,509,509
BEGIN DESCRIPTION:
CRYSTAL CREEK 50.0
END DESCRIPTION:
XS GIS Cut Line= 3
      3864117.82     10092811.07      3863347.29     10092757.45
      3861661.53     10093177.51
#Sta/Elev= 30
  4227.6  153.63  4267.7  152.47  4357.9  142.72    4408   140.3  4428.1  136.36
  4487.3  133.36  4688.7  127.44    4809  129.16    4839  127.15  4859.1  130.05
  4909.2  129.51 4936.16 126.227  4949.3  119.77  4996.4  115.19  5043.7  115.19
  5050.9     123    5082  126.39  5228.9  127.89  5408.8  125.14  5595.5  127.61
  5751.7  134.83  5903.4  131.17  6031.7  133.73  6133.1  131.24  6279.5  134.69
  6370.1  132.82    6438  134.37  6519.3  138.17  6687.2   149.9  6737.3  155.93
#Mann= 10 ,-1 , 0
  4227.6     .05       0  4487.3     .12       0 4936.16     .07       0
    5082      .1       0  5228.9     .12       0  5408.8      .1       0
  5595.5     .12       0  5903.4     .05       0    6438     .12       0
  6519.3     .05       0
Bank Sta=4936.16,5082
XS Rating Curve= 0 ,0
Exp/Cntr=0.3,0.1

Type RM Length L Ch R = 1 ,24515   ,515,515,515
BEGIN DESCRIPTION:
CRYSTAL CREEK 49.0
END DESCRIPTION:
XS GIS Cut Line= 3
      3864097.76     10092198.66      3863093.08       10092414.
      3861688.01     10092993.81
#Sta/Elev= 30
  3972.5  153.48    4154  147.42  4388.1  125.07  4785.3  125.88  4822.7  126.48
  4882.6  122.47  4933.8  124.41    4944  122.83  4960.7   115.7  4965.9  119.05
  4992.8     112  5040.1     112  5056.1   119.2  5061.5  114.78    5080  122.68
  5085.4  119.99    5103  125.17  5139.3  123.97    5228  123.51  5331.4  124.72
  5470.8  126.02    5530  129.59  5612.6  128.67    5698  132.68    5788  132.13
  5827.8  130.56  5926.8  132.69  6033.4   129.9  6163.7  131.46    6520  148.36
#Mann= 9 ,-1 , 0
  3972.5     .05       0    4154     .12       0  4785.3      .1       0
  4933.8     .07       0    5103      .1       0  5139.3     .12       0
    5228      .1       0  5331.4     .12       0    5788     .05       0
Bank Sta=4933.8,5103
XS Rating Curve= 0 ,0
Exp/Cntr=0.3,0.1

Type RM Length L Ch R = 1 ,24000   ,558,558,558
BEGIN DESCRIPTION:
CRYSTAL CREEK 48.0
END DESCRIPTION:
XS GIS Cut Line= 3
      3864017.83     10091861.07      3863240.43     10091962.57
      3861656.79     10092795.88
#Sta/Elev= 30
    4216  153.88  4255.7  153.02  4286.6  150.68  4316.8     143  4492.7  127.49
    4579  123.45  4656.8  124.52  4679.9  121.86  4700.1  124.94  4841.2  126.03
  4911.8   121.6  4941.3  125.78  4962.3   121.3  4968.9  112.31  5016.2  112.31
  5030.1  121.63  5090.1  122.36  5127.2  121.32  5140.3  126.15  5200.7  124.07
  5244.8  129.09    5534  131.14  5556.6  128.15  5756.7  125.55  6057.5  125.94
  6277.3  131.13  6411.9  129.82  6525.7  134.83  6598.6   140.1  6789.5  151.46
#Mann= 13 ,-1 , 0
    4216     .05       0  4255.7     .12       0  4492.7      .1       0
  4656.8     .12       0  4941.3      .1       0  4962.3     .07       0
  5030.1      .1       0  5090.1     .12       0  6057.5     .05       0
  6277.3     .12       0  6411.9     .05       0  6525.7     .12       0
  6598.6     .05       0
Bank Sta=4962.3,5030.1
XS Rating Curve= 0 ,0
Exp/Cntr=0.3,0.1

Type RM Length L Ch R = 1 ,23442   ,442,442,442
BEGIN DESCRIPTION:
CRYSTAL CREEK 47.0
END DESCRIPTION:
XS GIS Cut Line= 3
      3863337.35     10091261.15      3862813.82     10091771.47
      3861646.39     10092528.51
#Sta/Elev= 30
  4268.9  150.34  4501.9   142.3  4560.5  137.67  4671.6  132.09  4770.7   123.3
  4834.2  123.87  4855.4  115.16  4862.5  117.87  4869.5  112.91  4876.7  114.88
  4883.6  111.51  4890.8  117.07  4897.8     115    4905  118.98  4926.1  115.89
  4933.2  118.76  4940.2  115.97  4947.4  120.09  4995.3  110.31  5042.7  110.31
  5043.7  110.81  5046.3 120.083    5047  122.58  5152.9  125.12  5293.2  124.31
  5400.4  128.23  5698.4  123.12  5877.7  123.67  6095.3  133.14  6391.4  152.81
#Mann= 5 ,-1 , 0
  4268.9     .05       0  4560.5      .1       0  4947.4     .07       0
    5047      .1       0  5152.9     .12       0
Bank Sta=4947.4,5046.3
XS Rating Curve= 0 ,0
Exp/Cntr=0.3,0.1

Type RM Length L Ch R = 1 ,23000   ,500,500,500
BEGIN DESCRIPTION:
CRYSTAL CREEK 46.0
END DESCRIPTION:
XS GIS Cut Line= 3
      3863306.06     10091229.92      3862473.93     10091526.79
      3861629.04     10092174.33
#Sta/Elev= 30
  4116.5  150.88  4404.6   137.9  4422.5  139.34  4640.5  129.83  4845.5  126.03
  4868.4   123.2  4907.1  119.53  4912.4  116.64  4937.9  115.85  4943.2  111.88
  4963.4  112.37    4984  109.83  5031.4  109.83  5035.4  117.46  5049.9  121.36
  5064.5  119.54  5085.3  123.49    5185  118.76  5243.1  118.92  5263.9  122.75
  5384.7  120.64  5407.2  123.14  5442.5  122.45  5492.4  125.09  5572.9  122.69
    5655  123.06  5700.9  123.08    5809  129.05    5914  138.87  6064.5   149.2
#Mann= 8 ,-1 , 0
  4116.5     .05       0  4868.4     .07       0  5085.3     .05       0
  5384.7     .12       0  5572.9     .05       0    5655     .12       0
  5700.9     .05       0    5809     .12       0
Bank Sta=4868.4,5085.3
XS Rating Curve= 0 ,0
Exp/Cntr=0.3,0.1

Type RM Length L Ch R = 1 ,22500   ,500,500,500
BEGIN DESCRIPTION:
CRYSTAL CREEK 45.0
END DESCRIPTION:
XS GIS Cut Line= 3
      3863038.76     10090618.78      3862022.54     10091480.82
       3861458.9     10091684.76
#Sta/Elev= 30
  3667.4  151.85  3783.5  148.55  3904.3  141.28  4009.7  132.39    4102  127.87
  4364.5  125.52  4497.4   127.2  4571.1  126.92  4663.3  123.18  4802.9  123.52
  4946.7  120.75  4967.5  116.36  4972.4  108.15  5019.8  108.15  5020.8  108.65
  5026.3  120.48  5036.9  122.95  5068.8  120.83  5074.2  118.55  5079.5  120.67
  5090.1  117.36  5099.5  120.73  5136.1  122.82  5191.4  126.74  5216.8  126.38
  5278.1   131.9    5314  127.56    5370   128.4  5543.2  143.58  5599.4  145.85
#Mann= 6 ,-1 , 0
  3667.4     .12       0  4497.4     .05       0  4802.9      .1       0
  4946.7     .07       0  5026.3      .1       0  5136.1     .05       0
Bank Sta=4946.7,5026.3
XS Rating Curve= 0 ,0
Exp/Cntr=0.3,0.1

Type RM Length L Ch R = 1 ,22000   ,500,500,500
BEGIN DESCRIPTION:
CRYSTAL CREEK 44.0
END DESCRIPTION:
XS GIS Cut Line= 3
      3862717.82      10090211.1      3861916.81     10091039.73
      3861476.26     10091462.52
#Sta/Elev= 30
  3847.5  151.53  3943.3  146.87    4126  138.49  4335.3  126.19  4342.5  127.15
  4370.8  123.38  4469.9  121.09  4505.1  122.99  4519.3  121.75  4554.8  123.38
    4590  122.09  4618.3  124.73    4793  124.45  4887.1  119.62  4922.4  122.07
  4950.7  120.61  4957.9  114.02  4962.4  107.69  5009.9  107.69  5014.3   109.9
  5021.5   109.2  5028.4  112.27  5056.7  119.24    5085  120.17  5106.4  118.73
    5153  121.79  5247.9  131.74    5309  134.57  5337.2  135.32  5610.6  142.74
#Mann= 9 ,-1 , 0
  3847.5     .12       0  3943.3     .05       0    4126     .12       0
    4793      .1       0  4950.7     .07       0  5056.7      .1       0
    5153     .05       0    5309      .1       0  5337.2     .05       0
Bank Sta=4950.7,5056.7
XS Rating Curve= 0 ,0
Exp/Cntr=0.3,0.1

Type RM Length L Ch R = 1 ,21500   ,477,477,477
BEGIN DESCRIPTION:
CRYSTAL CREEK 43.0
END DESCRIPTION:
XS GIS Cut Line= 3
      3862524.85     10089986.85      3861817.11     10090592.03
      3861458.86     10091400.07
#Sta/Elev= 30
  4068.8  148.42  4093.5  146.93  4165.3  142.47  4348.7  135.02  4446.1  132.29
  4493.6   132.8  4608.5  131.12  4694.2  125.08  4735.9  120.18  4792.9  117.49
  4864.3  121.92  4899.8  121.72  4956.5  120.35  4970.8  115.42  4977.4  116.57
  4985.1  113.35  4989.2  107.44  5059.5  108.09    5065  112.37  5082.8  114.36
  5088.2  118.38  5108.8 120.675  5129.3  122.29  5181.3  119.93    5242  127.01
  5338.1  133.32  5476.5  137.63  5529.1  139.83  5726.2  139.11  5883.9  141.03
#Mann= 10 ,-1 , 0
  4068.8     .12       0  4093.5     .05       0  4165.3     .12       0
  4348.7     .05       0  4493.6     .12       0  4899.8      .1       0
  4956.5     .07       0  5108.8      .1       0    5242     .12       0
  5476.5     .05       0
Bank Sta=4956.5,5108.8
XS Rating Curve= 0 ,0
Exp/Cntr=0.3,0.1

Type RM Length L Ch R = 1 ,21023   ,523,523,523
BEGIN DESCRIPTION:
CRYSTAL CREEK 42.0
END DESCRIPTION:
XS GIS Cut Line= 3
      3862093.89     10089596.41      3861621.31     10090199.39
       3861431.1     10091292.36
#Sta/Elev= 30
  4233.9  138.26  4323.2  135.89  4381.7  133.84  4576.3  130.09  4646.8  124.98
  4661.3   125.4  4669.4  128.36  4739.9  124.14  4808.5  127.04  4847.5  126.71
  4897.2  112.16  4911.6  119.15  4929.8  119.76  4953.3  118.27  4967.7  112.27
  4972.7  106.67  5020.6  106.67  5021.6  107.17    5022  112.44  5048.4  117.99
    5141  118.57  5339.3  118.13  5377.3  123.83  5455.5  121.47  5549.8  123.24
  5862.7  136.27  5874.6  132.54  5884.8  132.61  5945.7  138.17  6109.4  139.99
#Mann= 9 ,-1 , 0
  4233.9     .05       0  4323.2     .12       0  4381.7     .05       0
  4808.5     .12       0  4929.8      .1       0  4953.3     .07       0
  5048.4     .05       0    5141      .1       0  5339.3     .05       0
Bank Sta=4953.3,5048.4
XS Rating Curve= 0 ,0
Exp/Cntr=0.3,0.1

Type RM Length L Ch R = 1 ,20500   ,500,500,500
BEGIN DESCRIPTION:
CRYSTAL CREEK 41.0
END DESCRIPTION:
XS GIS Cut Line= 3
      3861868.21     10089469.65      3861121.19     10090277.63
      3860581.67     10090538.32
#Sta/Elev= 30
  3899.6  143.26  4042.3  138.11  4155.7  128.53    4285  126.15  4538.4   121.2
    4588  120.74  4764.1  120.25  4863.3  116.41  4955.2   119.8  4969.4  118.11
  4976.7  113.58  4983.5  114.72    5000  105.67    5013  104.89  5060.9  104.89
  5070.6  108.94  5087.7   109.6  5093.2  115.25  5110.3  115.92  5115.8  119.59
    5161  118.25  5178.1  120.59  5223.3  107.18  5236.9  106.21  5251.4  107.45
  5281.4  118.87  5292.2  119.23  5454.8  133.07  5572.8  135.42  5599.2  135.33
#Mann= 8 ,-1 , 0
  3899.6     .05       0    4285     .12       0  4538.4     .05       0
    4588      .1       0  4955.2     .07       0  5115.8      .1       0
  5292.2     .05       0  5572.8     .12       0
Bank Sta=4955.2,5115.8
XS Rating Curve= 0 ,0
Exp/Cntr=0.3,0.1

Type RM Length L Ch R = 1 ,20000   ,500,500,500
BEGIN DESCRIPTION:
CRYSTAL CREEK 40.0
END DESCRIPTION:
XS GIS Cut Line= 3
       3861618.2      10089370.7      3860998.23     10089871.38
      3860140.49     10090427.04
#Sta/Elev= 30
  4203.1  143.33  4274.8  142.03  4367.5  133.81  4396.3  133.25  4452.3  127.69
  4524.2  124.32  4679.4  124.65  4778.2  122.68  4900.1  119.44  4936.2  117.12
  4938.3  115.31  4989.8  115.31    4997  116.76  5036.2  117.11  5058.9  119.61
  5064.9   119.3    5080  121.84  5131.5   125.7  5137.4  125.28  5143.4     127
  5192.6  127.83  5267.3  129.16  5359.6  128.93  5454.6  130.09  5500.1  129.14
  5587.9  130.93  5605.8  131.43  5817.3   130.3  5926.1  132.53    6022  132.71
#Mann= 8 ,-1 , 0
  4203.1     .05       0  4778.2     .12       0  4900.1     .07       0
  5058.9     .12       0  5192.6      .1       0  5359.6     .05       0
  5587.9     .12       0  5605.8     .05       0
Bank Sta=4900.1,5058.9
XS Rating Curve= 0 ,0
Exp/Cntr=0.3,0.1

Type RM Length L Ch R = 1 ,19500   ,500,500,500
BEGIN DESCRIPTION:
CRYSTAL CREEK 39.0
END DESCRIPTION:
XS GIS Cut Line= 3
      3861279.67      10089125.9      3860967.83     10089395.31
      3860097.38     10090381.11
#Sta/Elev= 30
  4587.9   147.4  4592.5  146.51  4600.2  146.72  4628.7  145.24  4635.3  144.21
  4656.4  143.72  4692.3  139.92  4720.8  138.71  4819.6  131.37  4827.2  131.35
  4876.6  125.82  4890.9   125.3  4897.5  125.99  4905.1  123.78  4911.7  123.94
  4919.4  121.87 4950.87  119.25  4968.8  118.23  4970.9  116.99  5022.4  116.99
  5032.7  119.29  5102.3  120.08    5149  120.62  5351.4  123.09  5379.9  122.87
  5517.8  125.17  5655.9  127.71  5883.2   127.9  6150.5  132.17  6315.1   133.1
#Mann= 9 ,-1 , 0
  4587.9     .12       0  4656.4     .05       0 4950.87     .05       0
  5032.7     .05       0  5102.3     .12       0    5149      .1       0
  5517.8     .05       0  5883.2     .12       0  6150.5     .05       0
Bank Sta=4950.87,5032.7
XS Rating Curve= 0 ,0
Exp/Cntr=0.3,0.1

Type RM Length L Ch R = 1 ,19000   ,500,500,500
BEGIN DESCRIPTION:
CRYSTAL CREEK 38.0
END DESCRIPTION:
XS GIS Cut Line= 3
      3860937.04     10088665.96      3860675.18     10089003.88
      3860051.64     10090348.21
#Sta/Elev= 30
  4572.5  146.84    4576  146.44  4582.3  146.95  4604.3  145.87  4611.3  144.49
  4654.8  139.67  4667.5  137.27  4696.4   133.4  4739.8  128.44  4754.3  127.51
  4799.4  122.61  4850.3  119.71  4889.2  119.22  4895.5  119.76  4924.5  120.08
  4959.8  118.37  4962.9  116.63  5014.7  116.63  5015.9  117.23  5032.4  118.01
  5215.6  119.87  5228.4  120.49  5263.9  120.88  5395.8   122.6  5579.6  124.94
  5780.9  127.46  5857.5  128.43  6078.9  131.32  6300.9  132.17  6481.9  133.59
#Mann= 11 ,-1 , 0
  4572.5     .12       0  4799.4      .1       0  4850.3     .12       0
  4924.5     .07       0  5228.4     .12       0  5263.9     .05       0
  5395.8      .1       0  5579.6     .12       0  5780.9     .05       0
  5857.5     .12       0  6300.9     .05       0
Bank Sta=4924.5,5228.4
XS Rating Curve= 0 ,0
Exp/Cntr=0.3,0.1

Type RM Length L Ch R = 1 ,18500   ,501,501,501
BEGIN DESCRIPTION:
CRYSTAL CREEK 37.0
END DESCRIPTION:
XS GIS Cut Line= 3
      3860618.89     10088433.45      3860386.03      10088607.3
      3859182.49     10089925.66
#Sta/Elev= 30
  4709.4  151.28  4759.2  147.66  4794.6  143.88  4800.8  142.55  4836.3  138.42
  4909.3     131  4931.9  126.91  4950.9  122.89  4965.5  116.15  4980.1  112.67
  4994.7   109.7  4995.4  104.89  4996.6  104.29  5048.4  104.29  5049.5  104.89
  5050.9  112.58  5058.3  113.08    5065  115.13  5079.2  117.81  5093.4  119.56
  5128.6  127.69    5136  127.83  5142.7  126.03  5150.2  125.82  5233.9  127.27
  5284.6  127.75  5659.6  116.82  6070.3  121.55  6197.4  121.35  6785.1  131.19
#Mann= 5 ,-1 , 0
  4709.4     .12       0  4931.9      .1       0  4980.1     .07       0
  5048.4      .1       0  5233.9     .05       0
Bank Sta=4980.1,5050.9
XS Rating Curve= 0 ,0
Exp/Cntr=0.3,0.1

Type RM Length L Ch R = 1 ,17999   ,499,499,499
BEGIN DESCRIPTION:
CRYSTAL CREEK 36.0
END DESCRIPTION:
XS GIS Cut Line= 3
      3860319.04     10088114.31      3859996.93     10088349.94
      3858839.62      10089466.9
#Sta/Elev= 30
  4606.1  144.31  4661.6  143.67  4676.3  141.64  4768.6  135.82  4797.5   134.3
  4805.8  135.15  4883.2  126.11  4891.7  124.07  4897.9  120.47  4912.5  118.29
  4918.7  114.05  4924.6  112.43 4930.47 109.347  4933.4  107.22  4941.9  106.24
  4948.1  103.63  4962.7  104.61  4965.8  102.69  5017.6  102.69  5018.7  103.29
  5019.4  108.01  5026.6  107.77  5033.5  109.52    5087  108.74  5281.3  108.12
  5373.9  109.58  5513.4  111.78  6228.7   123.1  6449.3  127.78  6613.6  130.61
#Mann= 8 ,-1 , 0
  4606.1     .12       0  4924.6      .1       0 4930.47     .07       0
  5033.5      .1       0    5087     .05       0  5373.9     .12       0
  5513.4     .05       0  6449.3     .12       0
Bank Sta=4930.47,5033.5
XS Rating Curve= 0 ,0
Exp/Cntr=0.3,0.1

Type RM Length L Ch R = 1 ,17500   ,500,500,500
BEGIN DESCRIPTION:
CRYSTAL CREEK 35.0
END DESCRIPTION:
XS GIS Cut Line= 3
      3860164.27     10087722.64      3859778.45     10088077.21
      3858524.98     10088742.96
#Sta/Elev= 30
    4476  141.58  4550.4  140.79  4592.9  138.45  4670.6   130.1    4805  121.31
  4811.8  119.37  4819.2  120.35    4826  116.88  4847.6  116.12  4868.6   118.6
  4875.9  116.89  4882.7  119.61  4911.1   119.3 4944.68 113.604  4953.6  110.82
  4974.6  108.94  4997.8  102.68  5068.6   103.6  5078.6  107.39  5084.2  105.71
  5100.5     114  5106.2  112.59  5122.5  114.04  5128.2  111.68  5172.2  116.23
  5238.5  115.98  5252.2  117.77  5321.8   119.9  6231.6  138.75  6419.3  140.09
#Mann= 5 ,-1 , 0
    4476     .12       0 4944.68     .07       0  5100.5      .1       0
  5252.2     .12       0  5321.8     .05       0
Bank Sta=4944.68,5100.5
XS Rating Curve= 0 ,0
Exp/Cntr=0.3,0.1

Type RM Length L Ch R = 1 ,17000   ,500,500,500
BEGIN DESCRIPTION:
CRYSTAL CREEK 34.0
END DESCRIPTION:
XS GIS Cut Line= 3
       3860096.6     10087563.04      3859429.65     10087765.12
      3858472.28     10088684.45
#Sta/Elev= 30
  4303.1  141.41  4386.6  136.91  4419.5  134.28  4447.2  130.04  4490.5  127.79
  4518.2  124.18  4636.2   116.4  4740.7  117.47  4803.3  114.89  4863.1  116.24
  4913.1  114.97  4934.1  116.59  4949.6   112.5  4960.1  111.91    4967  110.38
  4972.3  105.49    4981  105.07  4986.5  100.83  5038.7  100.83  5039.9  101.53
  5040.9  108.67  5055.1  112.14  5104.5  109.87    5140  119.76  5175.2  123.75
  5373.3  121.17  5408.6   128.1  5881.9  136.26    5953  136.83  6327.3  139.88
#Mann= 6 ,-1 , 0
  4303.1     .12       0  4913.1     .05       0  4960.1     .07       0
  5055.1     .05       0  5881.9     .12       0    5953     .05       0
Bank Sta=4960.1,5055.1
XS Rating Curve= 0 ,0
Exp/Cntr=0.3,0.1

Type RM Length L Ch R = 1 ,16500   ,624,624,624
BEGIN DESCRIPTION:
CRYSTAL CREEK 33.0
END DESCRIPTION:
XS GIS Cut Line= 3
       3860062.7     10087205.21      3859408.01     10087379.16
      3858152.77      10088138.4
#Sta/Elev= 30
  4322.6  140.25  4472.5  133.44  4544.9  124.98  4707.4  114.02  4824.3  111.59
  4917.4  116.15  4946.1  113.04  4951.3  114.78  4958.8  111.36  4986.3  102.52
  5046.5  103.55  5055.9  100.75  5108.1  100.75  5117.1  108.58  5126.1  112.23
  5131.9  106.74  5147.4  111.47  5153.3  108.59  5162.9  111.18  5168.8  107.36
  5175.5   111.9  5285.2  113.62  5300.7  118.22  5337.5  122.93  5512.1  119.94
  5777.6  120.29  6038.3  128.48    6295  134.62  6368.3  135.76    6467  137.39
#Mann= 8 ,-1 , 0
  4322.6     .12       0  4707.4      .1       0  4958.8     .07       0
  5126.1     .05       0  5777.6      .1       0  6038.3     .05       0
    6295     .12       0  6368.3     .05       0
Bank Sta=4958.8,5126.1
XS Rating Curve= 0 ,0
Exp/Cntr=0.3,0.1

Type RM Length L Ch R = 1 ,15876   ,656,656,656
BEGIN DESCRIPTION:
CRYSTAL CREEK 32.0
END DESCRIPTION:
XS GIS Cut Line= 3
       3859954.8     10086680.88      3859642.85     10086886.07
      3858019.08     10087865.74
#Sta/Elev= 30
  4644.6  151.97  4822.1  142.98  4880.3  135.66  4895.6  130.08  4924.6  118.97
  4952.2  112.41    4962  100.18  5014.2  100.18    5018  103.11  5047.2  109.08
  5082.2  112.17  5113.1  111.17  5134.6  113.93  5155.8  113.33  5186.8   116.4
    5214   114.3  5235.4     116  5252.5  115.18  5351.9  115.51  5382.9  119.13
  5388.7   118.3  5404.3  121.64  5410.1  119.72  5488.4  122.58  5536.3  124.12
  5664.2   123.4    6078  119.51  6222.8  118.75  6504.9  121.77  6914.4  137.19
#Mann= 10 ,-1 , 0
  4644.6     .12       0  4895.6     .05       0  4952.2     .05       0
  5082.2      .1       0  5134.6     .12       0  5252.5     .05       0
  5488.4    .075       0  5664.2     .05       0    6078     .12       0
  6222.8     .05       0
Bank Sta=4952.2,5082.2
XS Rating Curve= 0 ,0
Exp/Cntr=0.3,0.1

Type RM Length L Ch R = 1 ,15220   ,195,195,195
BEGIN DESCRIPTION:
CRYSTAL CREEK 31.0
END DESCRIPTION:
XS GIS Cut Line= 3
      3859790.76     10086009.55      3859378.43       10086367.
      3857853.58     10087686.36
#Sta/Elev= 30
  4454.3  147.82  4521.5  143.86  4542.4  146.23  4570.9  143.27    4606  144.63
    4776  140.45  4804.5  135.97  4812.1  131.73  4818.7  133.41  4826.4  130.24
  4840.6  131.28  4896.6  117.24  4932.7  121.46  4961.1  112.23  4961.5  100.54
  4962.6   99.84  5014.8   99.84  5045.7  110.71  5066.9  112.06  5102.8  110.96
  5123.6  114.63  5147.3  114.37  5232.4  114.26    5457  115.73  5563.4   121.5
  6151.3  121.27  6222.6  118.48  6357.5  122.03  6659.3  122.65  7016.4  131.97
#Mann= 6 ,-1 , 0
  4454.3     .05       0  4961.1     .03       0  5066.9     .05       0
  5147.3      .1       0  5232.4     .05       0  6659.3    .075       0
Bank Sta=4961.1,5066.9
XS Rating Curve= 0 ,0
Exp/Cntr=0.3,0.1

Type RM Length L Ch R = 1 ,15025   ,525,525,525
BEGIN DESCRIPTION:
CRYSTAL CREEK 30.0
END DESCRIPTION:
XS GIS Cut Line= 3
      3859662.93     10085892.02      3859220.69     10086255.74
      3857697.01     10087592.88
#Sta/Elev= 30
  4427.4   139.4  4778.6  124.63  4821.6  124.43  4848.9  119.98  4899.8  118.16
  4906.3  116.24  4920.7  117.99 4939.13 110.492  4949.4  105.03  4950.4   96.87
  4951.6   96.17    5004   96.17  5005.1   96.87  5005.5  100.73  5055.7  110.31
  5225.6  115.19  5799.7  116.56  5863.3   118.5  5884.2  121.98  5912.6  122.75
  5926.9  122.74  5955.3  117.52  5990.5  119.46  6012.3  123.81  6285.4  124.36
  6380.5  122.96  6617.8  124.52  6692.7   126.4    6855   129.2  7027.2  130.46
#Mann= 7 ,-1 , 0
  4427.4     .05       0 4939.13     .07       0  5055.7     .05       0
  6285.4    .075       0  6617.8     .05       0  6692.7    .075       0
    6855     .05       0
Bank Sta=4939.13,5055.7
XS Rating Curve= 0 ,0
Exp/Cntr=0.3,0.1

Type RM Length L Ch R = 1 ,14500   ,500,500,500
BEGIN DESCRIPTION:
CRYSTAL CREEK 29.0
END DESCRIPTION:
XS GIS Cut Line= 3
      3859434.79     10085684.36      3858858.02     10085891.07
      3857236.88     10086574.99
#Sta/Elev= 30
  4387.3  140.44  4490.3  140.14  4836.3  113.99  4936.4  112.52  4978.9  109.24
  4981.8   97.65    4983   96.95  5035.5   96.95  5038.4  102.66  5054.4  109.85
  5067.5  114.59  5091.2   111.9    5115  104.94  5120.4  107.73  5138.7  108.23
  5144.1  104.68  5162.4  108.59  5167.8  106.35  5191.5  111.24  5228.1  113.29
  5358.3  115.31  5390.9  118.44  5597.1  117.48  5694.8  120.94  5716.5  118.65
  5879.3   118.7  5933.6  123.82  5962.7     120    6053  118.91  6759.5  133.82
#Mann= 3 , 0 , 0
  4387.3     .05       0  4978.9     .07       0  5054.4     .05       0
Bank Sta=4978.9,5054.4
XS Rating Curve= 0 ,0
Exp/Cntr=0.3,0.1

Type RM Length L Ch R = 1 ,14000   ,500,500,500
BEGIN DESCRIPTION:
CRYSTAL CREEK 28.0
END DESCRIPTION:
XS GIS Cut Line= 3
      3859247.33     10085269.42      3858696.04     10085437.02
      3857148.38     10085644.42
#Sta/Elev= 30
  4423.8  142.64  4480.9  140.64  4611.4  130.84  4650.5   124.8  4759.5  118.04
 4815.04 111.879  4830.9   108.2  4858.1  108.68  4883.1   102.1    4904   104.3
  4935.4  100.82  4967.2  101.52  4972.1   96.43  5024.7   96.43  5048.6  108.43
  5058.7  111.89    5089  114.57  5119.2  115.23    5200  111.85  5310.9  110.53
  5421.9  117.47  5462.3  117.89  5512.7  116.21  5563.2  117.27  5591.8  115.76
  5643.9  119.44  5805.3  125.73  6037.4  124.96  6360.2  131.48  6561.5  133.09
#Mann= 3 , 0 , 0
  4423.8     .05       0 4815.04     .03       0  5058.7     .05       0
Bank Sta=4815.04,5058.7
XS Rating Curve= 0 ,0
Exp/Cntr=0.3,0.1

Type RM Length L Ch R = 1 ,13500   ,637,637,637
BEGIN DESCRIPTION:
CRYSTAL CREEK 27.0
END DESCRIPTION:
XS GIS Cut Line= 3
      3859247.34     10084868.37      3858500.92     10085039.56
      3857143.23     10085436.06
#Sta/Elev= 30
  4234.2  139.18  4267.4  137.84  4520.9  127.86    4562  124.21  4592.8  116.66
  4633.8  121.28  4718.5  112.93  4767.2  110.39  4847.2  111.91  4859.5  107.12
    4890  108.55  4895.2  104.96  4921.1  111.95  4938.1   112.3  4951.8  108.47
  4962.1  104.09  4972.7   95.57  5044.9   97.04  5054.5   99.26  5065.7  106.92
  5076.1  108.78  5107.4  107.94  5138.6  112.96  5211.5  109.08  5430.3  114.67
  5598.1   123.3  6008.2  127.12  6143.6  127.98    6320   132.9  6414.4  133.88
#Mann= 7 ,-1 , 0
  4234.2     .12       0  4267.4     .05       0  4951.8     .07       0
  5076.1     .05       0  6008.2     .12       0  6143.6     .05       0
    6320     .12       0
Bank Sta=4951.8,5076.1
XS Rating Curve= 0 ,0
Exp/Cntr=0.3,0.1

Type RM Length L Ch R = 1 ,12863   ,363,363,363
BEGIN DESCRIPTION:
CRYSTAL CREEK 26.0
END DESCRIPTION:
XS GIS Cut Line= 3
      3858950.43     10084394.42      3858168.21     10084524.73
      3857205.63     10084743.38
#Sta/Elev= 30
    4207  134.85  4281.8  133.58    4311  130.42  4403.5  125.45  4459.2   120.1
  4551.1  115.02  4574.6  113.77  4635.4  114.64  4878.7  112.53  4909.1   111.9
    4946  107.83  4966.9  107.44  4969.9  107.19  4980.1  104.64  4983.4   95.91
  4984.6   95.21  5037.3   95.21  5038.4   95.91  5041.4  104.95  5048.9  106.85
    5054  106.83  5072.1  112.61  5082.4  114.15  5173.9  116.62  5256.7  121.23
  5381.6  121.61  5505.3  123.27  5639.7  127.27  5768.9  127.77  5987.1   132.4
#Mann= 7 ,-1 , 0
    4207     .12       0  4551.1     .05       0  4966.9      .1       0
  4969.9     .07       0  5048.9      .1       0  5173.9     .12       0
  5381.6     .05       0
Bank Sta=4969.9,5048.9
XS Rating Curve= 0 ,0
Exp/Cntr=0.3,0.1

Type RM Length L Ch R = 1 ,12500   ,500,500,500
BEGIN DESCRIPTION:
CRYSTAL CREEK 25.0
END DESCRIPTION:
XS GIS Cut Line= 3
      3858929.59     10084097.55      3858218.27     10084177.53
      3857164.01       10084259.
#Sta/Elev= 30
  4284.2  137.07  4406.7  134.62    4451  132.13  4567.7  122.37  4649.9  113.37
  4716.1  110.85  4748.8  112.15  4832.5  111.56  4859.5  111.98  4879.7  107.78
    4930  111.59  4950.1  110.33  4958.6   95.44  4959.8   94.74  5012.5   94.74
  5030.5   96.59  5060.6  109.72  5160.9  115.58    5191  115.81    5211  114.01
  5240.9   114.8  5301.3  116.16  5321.4  118.59  5481.8  118.42  5552.1  122.06
  5612.2  122.01  5652.7  123.89  5722.6  126.16  5888.8  126.16  6057.4  129.46
#Mann= 7 ,-1 , 0
  4284.2     .12       0  4649.9     .05       0  4832.5      .1       0
  4950.1     .07       0  5060.6      .1       0  5240.9     .12       0
  5652.7     .05       0
Bank Sta=4950.1,5060.6
XS Rating Curve= 0 ,0
Exp/Cntr=0.3,0.1

Type RM Length L Ch R = 1 ,12000   ,500,500,500
BEGIN DESCRIPTION:
CRYSTAL CREEK 24.0
END DESCRIPTION:
XS GIS Cut Line= 3
      3858861.96     10083740.77      3858177.03     10083688.75
      3857312.63     10083944.71
#Sta/Elev= 30
  4313.1  137.83    4510  134.81    4578  131.29  4636.2  121.69  4718.4  111.31
  4778.5  106.41  4798.6  107.42  4838.7  105.61  4879.6  110.15  4918.9  108.51
    4939   110.8    4949  109.54  4969.1  103.15  4969.5   96.82  4970.7   96.12
  5023.4   96.12  5025.5   98.38  5040.9   97.86  5051.3   103.2  5082.6  105.14
  5097.2  109.62  5103.4  113.08  5159.5  110.57  5301.6   118.2  5437.2  118.33
  5588.9  123.31  5715.9  122.96  5765.6  125.15    5823  123.89  5901.5  126.22
#Mann= 6 ,-1 , 0
  4313.1     .12       0  4879.6      .1       0    4949     .07       0
  5097.2      .1       0  5159.5     .12       0  5715.9     .05       0
Bank Sta=4949,5097.2
XS Rating Curve= 0 ,0
Exp/Cntr=0.3,0.1

Type RM Length L Ch R = 1 ,11500   ,500,500,500
BEGIN DESCRIPTION:
CRYSTAL CREEK 23.0
END DESCRIPTION:
XS GIS Cut Line= 3
      3858892.26     10083354.48      3858108.25     10083213.41
      3857370.08      10083726.9
#Sta/Elev= 30
  4203.4  135.22  4319.6  133.55  4390.8  128.84  4471.8   119.4  4624.5   110.2
  4689.3  108.69  4782.9  108.63  4867.6  109.16  4926.3  111.44  4949.6  107.64
  4958.7    94.9  5011.4    94.9  5012.6    95.6  5012.7    97.1  5062.3   96.72
  5077.2   99.23  5085.8  102.95    5092  108.02  5098.1  106.82  5106.9  109.57
  5149.6  110.46  5207.6   109.6  5342.5  118.38  5414.7  120.82  5500.5  121.12
    5566  123.44  5595.7   122.2  5646.1  123.52    5703  121.55  5899.2  124.16
#Mann= 7 ,-1 , 0
  4203.4     .05       0  4471.8     .12       0  4689.3      .1       0
  4782.9     .12       0  4949.6     .07       0    5092     .12       0
  5149.6     .12       0
Bank Sta=4949.6,5092
XS Rating Curve= 0 ,0
Exp/Cntr=0.3,0.1

Type RM Length L Ch R = 1 ,11000   ,500,500,500
BEGIN DESCRIPTION:
CRYSTAL CREEK 22.0
END DESCRIPTION:
XS GIS Cut Line= 3
      3858931.36     10083263.33      3858236.11     10082755.79
      3857585.84     10082512.46
#Sta/Elev= 30
  4139.2  133.99  4286.6  128.44  4336.8  121.63  4372.3  121.13  4378.8  119.12
  4401.6  119.12  4487.4  113.13  4508.2  111.67  4552.1  112.91    4594  109.18
  4614.8   112.3  4644.2  113.09  4778.7  112.41  4858.3  109.08    4874  108.53
    4916  104.37  4930.7   99.93  4936.9  102.24  4945.4   98.65  4973.2   94.01
  5026.4   94.01  5027.6   94.71  5031.6  106.83  5040.8  108.83  5066.9  111.35
  5158.3  107.36  5197.3  112.34  5288.1  114.17  5415.5  122.33  5694.3  124.31
#Mann= 8 ,-1 , 0
  4139.2     .05       0  4487.4     .12       0  4778.7      .1       0
  4858.3     .05       0    4874     .07       0  5040.8      .1       0
  5066.9     .12       0  5415.5     .05       0
Bank Sta=4874,5040.8
XS Rating Curve= 0 ,0
Exp/Cntr=0.3,0.1

Type RM Length L Ch R = 1 ,10500   ,500,500,500
BEGIN DESCRIPTION:
CRYSTAL CREEK 21.0
END DESCRIPTION:
XS GIS Cut Line= 3
      3859043.15      10082094.6      3858343.53     10082301.95
      3857616.29     10082395.28
#Sta/Elev= 30
  4270.3  139.04  4432.3  132.44  4589.1  115.74  4659.6  108.54  4664.8  106.89
  4682.6  107.83  4693.2  104.61  4703.5   101.6  4745.2  108.54  4797.2  110.79
  4836.2  110.39  4901.6  112.91  4946.3   110.6  4964.2  104.17  4974.4   99.14
  4979.1   94.62  5032.4   94.62  5036.7   96.88  5111.3  103.94  5126.7  105.15
  5207.9  102.93  5270.5  104.19  5318.3  100.37    5345  102.62  5350.1  101.75
  5388.8  111.97  5479.6  119.45  5579.5  123.63    5651  125.57  5733.2  125.19
#Mann= 8 ,-1 , 0
  4270.3     .12       0  4589.1     .05       0  4693.2      .1       0
  4797.2     .05       0  4964.2     .03       0  5111.3      .1       0
  5207.9     .12       0  5579.5     .05       0
Bank Sta=4964.2,5111.3
XS Rating Curve= 0 ,0
Exp/Cntr=0.3,0.1

Type RM Length L Ch R = 1 ,10000   ,500,500,500
BEGIN DESCRIPTION:
CRYSTAL CREEK 20.0
END DESCRIPTION:
XS GIS Cut Line= 3
      3858859.83     10081651.28      3858236.71     10081863.58
      3857622.75     10082176.06
#Sta/Elev= 30
  4341.7  135.82  4534.3  129.75  4650.2  120.82  4713.5  112.69  4755.1  109.56
    4872  106.29  4903.7  107.23  4917.1  105.53  4943.2   96.56  4974.5   95.86
  4977.6   93.83  5032.2   93.83  5049.4  100.21    5055    99.2    5066  102.66
  5071.6  101.11  5077.3  104.92  5088.3  107.86  5090.3  107.57  5110.5  106.31
  5132.8  108.65    5167  109.11  5177.2  107.81    5200  107.92  5294.1  109.87
    5369  116.64  5427.5  117.23  5466.4  121.37  5533.2  124.98  5688.9  124.74
#Mann= 7 ,-1 , 0
  4341.7     .12       0  4534.3     .05       0  4903.7     .07       0
  5088.3     .05       0  5090.3     .12       0  5177.2      .1       0
    5200     .12       0
Bank Sta=4903.7,5088.3
XS Rating Curve= 0 ,0
Exp/Cntr=0.3,0.1

Type RM Length L Ch R = 1 ,9500    ,500,500,500
BEGIN DESCRIPTION:
CRYSTAL CREEK 19.0
END DESCRIPTION:
XS GIS Cut Line= 3
      3858818.17     10081375.23      3858141.73     10081390.18
      3857245.27      10081729.4
#Sta/Elev= 30
  4323.4  130.33  4443.7  125.21  4543.8  116.97  4613.8  113.37  4703.8  106.65
  4743.8  105.79  4768.4  107.21  4843.8  109.68  4881.6     108  4913.9  106.44
  4943.9   96.78  4963.9   95.43  4972.1   93.35  5026.7   93.35  5036.2  100.71
  5043.2  104.11  5048.6   103.5  5057.6  106.31    5070  108.62  5098.2  110.47
  5177.1   111.4  5207.3  112.83  5250.1   112.6  5323.5  116.76  5401.5  119.15
  5506.7  119.65  5592.2  116.78  5763.3   115.4    5913  120.73  5958.5  120.19
#Mann= 8 ,-1 , 0
  4323.4     .12       0  4768.4      .1       0  4881.6     .05       0
  4913.9     .07       0  5057.6      .1       0    5070     .12       0
  5177.1     .05       0  5401.5     .12       0
Bank Sta=4913.9,5057.6
XS Rating Curve= 0 ,0
Exp/Cntr=0.3,0.1

Type RM Length L Ch R = 1 ,9000    ,500,500,500
BEGIN DESCRIPTION:
CRYSTAL CREEK 18.0
END DESCRIPTION:
XS GIS Cut Line= 3
      3859109.87     10080812.73      3858273.76     10080910.52
      3857121.56     10081431.95
#Sta/Elev= 30
  4158.2  129.59  4260.9  123.19    4422  109.31    4573  108.93  4643.5  106.45
  4667.7  108.03  4744.2  108.53  4814.7  104.05  4885.1  107.17  4915.3  105.96
  4955.6   99.92  4961.2   96.06  4966.2   95.68  4968.1   92.46  5022.8   92.46
  5035.8    96.4  5041.3   95.38  5058.9  103.58  5087.5  107.19    5089  107.11
  5116.3  105.27    5215  111.43  5309.4  111.57  5555.3  118.19  5659.8  117.44
  5770.5  112.71  5934.6  114.73  5994.4  113.48  6190.8   121.2  6264.7  120.85
#Mann= 9 ,-1 , 0
  4158.2     .12       0  4667.7     .05       0  4885.1     .07       0
  5087.5     .05       0    5089     .12       0  5309.4     .05       0
  5659.8     .12       0  5770.5     .05       0  6190.8     .12       0
Bank Sta=4885.1,5087.5
XS Rating Curve= 0 ,0
Exp/Cntr=0.3,0.1

Type RM Length L Ch R = 1 ,8500    ,500,500,500
BEGIN DESCRIPTION:
CRYSTAL CREEK 17.0
END DESCRIPTION:
XS GIS Cut Line= 3
      3858984.88     10080250.23      3858249.58     10080414.83
      3856927.81     10081026.17
#Sta/Elev= 30
  4246.5  138.82  4397.2  128.16  4498.3  125.63  4595.3  118.14  4632.9  117.45
  4643.9  113.28  4745.6  103.87  4779.1   103.7  4822.5  107.64  4919.9   103.5
  4940.3  105.02  4957.8  100.31  4962.9  102.05  4981.3   96.33  5023.7   92.25
  5078.4   92.25    5090     102  5102.4  105.27  5112.1  107.37  5165.7  106.52
  5252.4  109.42  5349.6  110.43  5585.8  108.73  5835.2  113.44  6121.4   113.1
  6195.7  117.64  6247.1  116.55  6346.1  120.79  6384.6   119.9  6456.3  123.95
#Mann= 6 ,-1 , 0
  4246.5     .12       0  4919.9      .1       0  4940.3     .07       0
  5102.4      .1       0  5252.4     .12       0  5349.6     .05       0
Bank Sta=4940.3,5102.4
XS Rating Curve= 0 ,0
Exp/Cntr=0.3,0.1

Type RM Length L Ch R = 1 ,8000    ,500,500,500
BEGIN DESCRIPTION:
CRYSTAL CREEK 16.0
END DESCRIPTION:
XS GIS Cut Line= 3
      3858760.96     10079692.92      3858080.32     10079946.95
      3856872.08     10080915.46
#Sta/Elev= 30
  4273.5  135.64  4436.9   137.4  4671.7  130.67  4740.6  123.84  4765.6  124.61
  4820.9  121.65  4842.5  119.03  4851.2   114.5  4863.9  104.05  4874.5  101.55
  4911.5  102.62  4949.3  102.34  4959.9  100.12  4963.3   93.02  4964.6   92.22
  5019.4   92.22  5047.3    98.5  5054.4  102.32  5061.7  105.88    5078  107.52
  5192.4  106.87  5196.2  106.87    5353  111.09  5496.5  107.65  5751.5  108.02
  5865.1  112.05  6042.8  111.28  6306.8  119.94  6519.7  123.43  6548.5  121.84
#Mann= 8 ,-1 , 0
  4273.5     .12       0  4911.5      .1       0  4949.3     .07       0
  5054.4      .1       0    5078     .12       0  5192.4      .1       0
  5196.2     .12       0  5496.5     .05       0
Bank Sta=4949.3,5054.4
XS Rating Curve= 0 ,0
Exp/Cntr=0.3,0.1

Type RM Length L Ch R = 1 ,7500    ,500,500,500
BEGIN DESCRIPTION:
CRYSTAL CREEK 15.0
END DESCRIPTION:
XS GIS Cut Line= 3
      3858229.64     10079239.83      3857763.83     10079583.38
      3856667.16     10080614.82
#Sta/Elev= 30
  4421.2  131.93    4817  125.68  4881.8  121.89  4903.4  117.73  4917.3  114.91
  4938.1  104.95  4952.7   95.83  4953.3   92.74  4954.6   91.94  5009.4   91.94
    5031   94.84  5037.8   99.02  5080.3  104.95  5101.8  103.03  5158.4  105.29
  5200.5  109.49  5238.7  109.49  5306.9  107.31  5397.6  108.97  5439.2  108.11
  5535.5  104.98  5561.4  103.54  5575.5   106.6  5646.4  109.61    5724  108.29
  5759.7  111.72  5794.8  109.53  5978.9  111.28  6134.3  116.89  6505.5  123.82
#Mann= 8 ,-1 , 0
  4421.2     .12       0  4903.4      .1       0  4938.1     .07       0
  5080.3      .1       0  5238.7     .12       0  5397.6     .05       0
  5439.2     .12       0  5535.5     .05       0
Bank Sta=4938.1,5080.3
XS Rating Curve= 0 ,0
Exp/Cntr=0.3,0.1

Type RM Length L Ch R = 1 ,7000    ,500,500,500
BEGIN DESCRIPTION:
CRYSTAL CREEK 14.0
END DESCRIPTION:
XS GIS Cut Line= 3
      3858068.24     10078857.85      3857400.76     10079244.74
      3856599.44     10080552.34
#Sta/Elev= 30
  4228.5  128.96  4384.7  119.62    4422  115.31  4836.8  107.59  4888.3   104.4
  4910.9  106.14  4925.6  102.64  4957.1    94.9  4986.8    93.1  5041.6    93.1
  5050.9  103.28  5078.1   106.8    5109  103.62  5124.4  107.04  5239.1  106.96
  5264.9  107.51  5319.8  104.55  5429.6  104.61  5457.1  102.08  5631.2  110.48
  5973.5  110.05  6004.3  113.79  6031.6  110.33  6147.6  110.49  6163.1  113.54
  6184.4   111.9  6199.8  115.16  6250.6  115.12  6285.8  118.28  6533.6  124.18
#Mann= 6 ,-1 , 0
  4228.5     .12       0  4836.8      .1       0  4925.6     .07       0
  5050.9      .1       0  5239.1     .12       0  5264.9     .05       0
Bank Sta=4925.6,5050.9
XS Rating Curve= 0 ,0
Exp/Cntr=0.3,0.1

Type RM Length L Ch R = 1 ,6500    ,500,500,500
BEGIN DESCRIPTION:
CRYSTAL CREEK 13.0
END DESCRIPTION:
XS GIS Cut Line= 3
      3858120.28     10078519.33       3857198.5     10078795.26
      3856480.96     10080544.41
#Sta/Elev= 30
  4037.8  128.61  4339.1  118.37    4515  107.61  4548.1   101.8  4614.2  101.93
  4666.6   106.1  4758.4  105.51  4795.4  105.79  4823.2   98.36  4875.4  103.74
  4899.9   99.33  4948.5   99.46  4952.4   92.09  5060.3   94.09  5090.6   99.18
  5103.6  106.48    5128  106.56  5154.8  104.79    5363  105.69  5405.5   98.86
  5477.9  103.55  5698.8  107.12  5946.6  110.44  6314.1  109.78  6346.6     114
    6379  110.85  6530.3  110.66  6568.8  115.19  6622.2  112.46  6890.6  125.05
#Mann= 8 ,-1 , 0
  4037.8     .12       0  4758.4      .1       0  4948.5     .07       0
  5090.6      .1       0    5128     .12       0  5154.8      .1       0
  5477.9     .12       0  5698.8     .05       0
Bank Sta=4948.5,5090.6
XS Rating Curve= 0 ,0
Exp/Cntr=0.3,0.1

Type RM Length L Ch R = 1 ,6000    ,500,500,500
BEGIN DESCRIPTION:
CRYSTAL CREEK 12.0
END DESCRIPTION:
XS GIS Cut Line= 4
      3858165.84     10078280.61       3857365.4     10078330.62
      3857035.66     10078686.64      3856383.99     10080536.76
#Sta/Elev= 30
    4198  127.17  4762.8  104.24  4787.1  102.22  4827.2  106.91  4867.3  100.77
  4887.3  104.67    4918  103.86  4929.7  101.54  4947.4   93.95  5020.7   92.34
  5075.6   92.34  5083.3   97.91  5111.6  101.52  5207.9   105.2  5238.1  105.45
  5324.2  105.86  5373.6   99.47  5527.6  105.06  5669.6   95.95  5762.5   98.66
  5767.8  101.76  5793.4   99.03  5798.7  103.27  5824.4  101.78  5829.7   107.4
  6176.5  111.19  7101.5  108.97  7296.9  116.39  7308.2  116.56  7446.8  127.36
#Mann= 11 ,-1 , 0
    4198     .12       0  4762.8     .05       0    4918      .1       0
  4929.7     .07       0  5111.6      .1       0  5207.9     .12       0
  5238.1      .1       0  5527.6     .12       0  6176.5     .05       0
  7296.9     .12       0  7308.2     .05       0
Bank Sta=4929.7,5111.6
XS Rating Curve= 0 ,0
Exp/Cntr=0.3,0.1

Type RM Length L Ch R = 1 ,5500    ,1000,1000,1000
BEGIN DESCRIPTION:
CRYSTAL CREEK 11.0
END DESCRIPTION:
XS GIS Cut Line= 4
      3858117.81     10078061.06      3857453.96     10077838.73
      3856418.47     10078495.78      3856307.36     10080592.98
#Sta/Elev= 30
  4299.9  126.18  4574.1  113.59    4726  110.78  4826.8  103.72  4852.2  103.08
  4869.3   97.95  4890.4  100.71  4922.1   97.41  4926.3    91.6  4981.2    91.6
  5028.7   95.49  5042.8   93.58 5049.34  97.467  5107.5   96.71  5137.5  104.48
  5237.9   100.8  5469.1  108.26  5869.1  104.52  6150.6  106.71  6622.2  103.71
  6692.3  107.11  6892.6  109.15  7543.5  108.25  7741.9  110.69  7880.2  109.53
  8054.2  109.29    8135  112.76  8233.3  121.56  8264.5  120.15  8326.5  127.23
#Mann= 9 ,-1 , 0
  4299.9     .12       0  4826.8     .05       0  4922.1     .03       0
 5049.34     .12       0  6150.6     .05       0  7741.9      .1       0
  7880.2     .05       0    8135     .12       0  8233.3     .05       0
Bank Sta=4922.1,5049.34
XS Rating Curve= 0 ,0
Exp/Cntr=0.3,0.1

Type RM Length L Ch R = 1 ,4500    ,1000,1000,1000
BEGIN DESCRIPTION:
CRYSTAL CREEK 9.0
END DESCRIPTION:
XS GIS Cut Line= 3
      3858404.61     10077599.96      3857361.16     10076905.35
      3848611.82     10078053.87
#Sta/Elev= 30
  3746.5  133.17    4782   104.7    4974   94.52  5086.3   96.92  5266.6   101.7
  5768.6  103.82  6380.6  102.61  6486.5  103.58  6747.2  102.82  7037.4  103.83
  7262.6  106.81  7302.9   96.61    7305   83.49  7307.3   80.69  7618.4   83.49
    7901    83.7  8755.3   85.31  8795.6   98.56  9239.4  101.33 10979.7      96
 11100.7   93.62 11300.6  100.52 11382.6    86.8 11600.6   86.63 11791.1   87.35
 11871.8  103.58 12753.7  103.23 13000.5  103.14 13268.8  107.33 13824.4  118.83
#Mann= 20 ,-1 , 0
  3746.5     .12       0    4782     .05       0    4974      .1       0
  5086.3     .12       0  5266.6     .05       0  5768.6     .12       0
  6380.6     .12       0  6486.5      .1       0  6747.2     .12       0
  7037.4     .05       0    7305     .03       0  7618.4     .05       0
    7901      .1       0 10979.7      .1       0 11100.7     .12       0
 11300.6     .05       0 11600.6     .12       0 12753.7      .1       0
 13000.5     .12       0 13268.8     .05       0
Bank Sta=7305,7618.4
XS Rating Curve= 0 ,0
Exp/Cntr=0.3,0.1

Type RM Length L Ch R = 1 ,3500    ,1213,1213,1213
BEGIN DESCRIPTION:
CRYSTAL CREEK 7.0
END DESCRIPTION:
XS GIS Cut Line= 3
      3858694.86      10077354.9      3857211.52     10075932.96
      3849687.12     10074130.41
#Sta/Elev= 30
  2945.2  127.49  3221.6  106.82  4200.7  103.97  4770.4  100.01  4811.8   81.89
  4814.1   79.09  5125.2   81.89  5137.5   96.97  5155.6   99.01  5313.8  100.18
  6318.9  102.26  6751.9  100.64  6788.7   87.01  6817.1   84.16  7121.8   82.77
  7183.8   94.33  7324.1   97.18  7625.7   91.81  7733.8   91.36  7769.9  101.87
    7811  104.24  8118.2  101.56  8932.4  100.78  9032.9  100.66 10319.8  103.01
 11210.1   110.5 11841.9  108.46 12249.5  116.27 12410.6  117.84 12737.3  117.31
#Mann= 16 ,-1 , 0
  2945.2     .12       0  4200.7     .05       0  4811.8     .03       0
  5125.2    .075       0  5313.8     .12       0  6318.9      .1       0
  6817.1     .05       0  7121.8      .1       0  7324.1     .05       0
  7625.7      .1       0  8118.2     .05       0  8932.4     .12       0
  9032.9      .1       0 10319.8     .05       0 12249.5    .075       0
 12410.6     .05       0
Bank Sta=4811.8,5125.2
XS Rating Curve= 0 ,0
Exp/Cntr=0.3,0.1

Type RM Length L Ch R = 1 ,2287    ,784,784,784
BEGIN DESCRIPTION:
CRYSTAL CREEK 5.0
END DESCRIPTION:
XS GIS Cut Line= 4
      3859043.22      10077246.9       3857003.3      10075285.1
      3856419.85     10075194.01      3849694.03      10073942.9
#Sta/Elev= 30
  1579.3  120.47  1874.1  108.49  2265.4  104.87  2888.8   114.5  3184.3  105.66
  3775.1  105.05  4295.9   125.6  4454.8  103.31  4819.8   98.85  4883.8   81.31
  4886.1   78.51  5197.2   81.31  5203.9   102.6  5479.3  101.02  5679.8   97.82
  6077.1  101.28  6328.2    85.2  6375.2   98.06  6426.1    83.8  6674.9   90.51
  6973.8  102.18    7911  103.58  8094.2  120.84  8134.9  106.33    8269  108.42
  8761.1  116.04  8910.5  102.93  9464.5  100.29 11553.3  116.13 11841.2  118.67
#Mann= 20 ,-1 , 0
  1579.3     .12       0  1874.1     .05       0  2265.4     .12       0
  2888.8     .05       0  3184.3    .075       0  3775.1     .05       0
  4454.8     .05       0  4883.8     .03       0  5197.2     .05       0
  5479.3    .075       0  5679.8    .075       0  6077.1     .05       0
  6328.2      .1       0  6674.9     .12       0  6973.8     .05       0
    7911    .075       0    8269     .05       0  8910.5      .1       0
  9464.5     .05       0 11553.3     .05       0
Bank Sta=4883.8,5197.2
XS Rating Curve= 0 ,0
Exp/Cntr=0.3,0.1

Type RM Length L Ch R = 1 ,1503    ,1003,1003,1003
BEGIN DESCRIPTION:
CRYSTAL CREEK 3.0
END DESCRIPTION:
XS GIS Cut Line= 4
      3859268.92     10077055.94      3856617.86      10074484.7
      3854048.22     10074005.41      3849735.69     10073672.07
#Sta/Elev= 30
  1222.5  114.68  1786.4  109.16  2227.5  100.79  3403.7   99.06  4663.7  109.08
  5084.9   83.61  5210.7   83.25  5261.5   97.86    5587   87.65    6220   99.66
  6238.1   98.67  6254.3   76.21  6256.5   73.41  6565.5   73.41  6567.8   76.21
  6665.3   93.67  7420.1   88.53  8053.4   97.42  8560.4   99.35  8743.9   98.08
  8941.2   98.25  9340.7   99.27  9636.2  102.32 10026.3  104.64   10218  105.78
 10420.9  106.99 10716.9  109.41   11191  117.61 11407.4  118.69   11855  118.95
#Mann= 20 ,-1 , 0
  1222.5     .12       0  1786.4    .075       0  2227.5     .05       0
  3403.7     .05       0  5084.9      .1       0  6254.3     .03       0
  6565.5      .1       0  7420.1      .1       0  8053.4     .05       0
  8560.4    .075       0  8743.9     .05       0  8941.2    .075       0
  9340.7     .05       0  9636.2      .1       0 10026.3     .05       0
   10218    .075       0 10420.9     .12       0 10716.9    .075       0
   11191    .075       0 11407.4     .05       0
Bank Sta=6254.3,6567.8
XS Rating Curve= 0 ,0
Exp/Cntr=0.3,0.1
