HEC-RAS study STEWARTS CREEK.prj: STEWARTS CREEK Base Level Engineering

--- STEWARTS CREEK.g01 (geometry) --- (continued)

Type RM Length L Ch R = 1 ,83500   ,74,74,74
BEGIN DESCRIPTION:
STEWARTS CREEK 164.0
END DESCRIPTION:
XS GIS Cut Line= 3
      3823987.95     10138254.22      3824067.41     10136876.81
      3823817.85     10136011.06
#Sta/Elev= 30
  3620.3  289.88    3884  285.79    3944  282.62  4004.1  280.87  4144.3  278.93
  4229.6  276.25  4324.6   272.6  4444.8  271.37  4525.4  268.71  4595.1  268.15
  4643.5  269.99  4655.2  270.25  4675.2  268.97  4685.2  267.55  4721.1   266.4
  4765.3  267.43  5164.1  266.98  5192.5  267.29  5203.7  269.22  5224.5  273.02
  5245.3  274.73  5349.4  275.34  5376.5  276.52  5422.3  276.34  5474.3  274.57
  5578.4  276.56  5627.7  279.29  5733.9  283.13    5778  286.68    5901  292.24
#Mann= 6 ,-1 , 0
  3620.3     .11       0  4229.6     .17       0  4525.4     .11       0
  4643.5     .17       0  4675.2     .04       0  5203.7     .11       0
Bank Sta=4675.2,5203.7
XS Rating Curve= 0 ,0
Exp/Cntr=0.3,0.1

Type RM Length L Ch R = 1 ,83426   ,83,83,83
BEGIN DESCRIPTION:
Mapping XS 5d8391e6
END DESCRIPTION:
XS GIS Cut Line= 3
      3824086.04     10138260.79      3824141.05     10136877.79
      3823960.54     10136014.25
#Sta/Elev= 30
  3615.9  286.27  3805.8  286.93    4136  279.62    4272  275.21  4376.2   271.1
  4652.3  264.75  4716.5  270.58  4756.5  267.24  4896.6  267.57  4916.6  270.67
  4926.7  270.68  4946.7  268.06    5000  267.22  5027.3   260.5  5098.8   260.5
  5129.5  267.08  5170.3  268.12 5178.27  270.64  5186.2  272.63  5236.1  273.91
  5262.3  276.03  5336.1  275.66    5381  274.04    5436  274.63  5530.9  273.38
  5575.8  276.36  5630.8   277.6  5691.3  281.01  5820.5  283.44  5882.2  285.93
#Mann= 4 ,-1 , 0
  3615.9     .11       0    4272     .11       0  4926.7     .04       0
 5178.27     .11       0
Bank Sta=4926.7,5178.27
XS Rating Curve= 0 ,0
Exp/Cntr=0.3,0.1

Type RM Length L Ch R = 1 ,83343   ,245,245,245
BEGIN DESCRIPTION:
STEWARTS CREEK 163.0
END DESCRIPTION:
XS GIS Cut Line= 3
      3824159.83     10138247.71      3824216.75     10136845.56
      3824072.06     10136014.77
#Sta/Elev= 30
  3596.7  285.52  3973.6   283.4  4243.9  276.75    4384  269.43    4410  268.94
    4415  271.07  4594.2  264.29  4674.2  264.61  4704.2  262.44  4734.3  264.61
  4754.8  263.42    4853   263.9  4901.7  264.69  4906.7  262.06  4930.3  260.07
  4938.6  260.07  4944.4  262.97  4964.5  261.26  5014.7  262.25  5026.3  264.47
  5045.2   267.1  5080.8  267.92  5085.9  270.06  5135.4  270.13  5259.6  274.45
  5433.3  271.95  5552.7  277.63    5644  276.33  5726.2  279.37  5843.3  280.61
#Mann= 5 ,-1 , 0
  3596.7     .11       0  4754.8     .17       0    4853     .11       0
  4901.7     .04       0  5026.3     .11       0
Bank Sta=4901.7,5026.3
XS Rating Curve= 0 ,0
Exp/Cntr=0.3,0.1

Type RM Length L Ch R = 1 ,83098   ,196,196,196
BEGIN DESCRIPTION:
Mapping XS 729ab2d8
END DESCRIPTION:
XS GIS Cut Line= 3
      3824399.53     10137885.62        3824461.     10136866.35
      3824511.35     10136095.52
#Sta/Elev= 30
  3980.3  283.06    4065   282.6  4225.3   277.8  4255.3  277.81  4305.4  274.84
  4385.6  273.26    4616  264.99  4695.5  266.27  4756.3  264.58  4816.4   261.4
  4846.4  260.94  4863.8  262.02  4868.8  261.35  4896.5  262.55  4926.6  262.18
  4936.6  262.88  4956.6  261.22  4982.4  257.76  5006.7  258.54 5021.19261.2125
  5056.8  262.61  5106.9  261.14    5147  261.13  5379.9  274.14  5433.2  275.97
  5567.9  279.22  5577.9  278.67  5638.1  279.45  5688.9  282.01  5773.9  283.48
#Mann= 6 ,-1 , 0
  3980.3     .11       0  4956.6     .04       0 5021.19     .11       0
  5379.9    .125       0  5433.2     .11       0  5688.9    .125       0
Bank Sta=4956.6,5021.19
XS Rating Curve= 0 ,0
Exp/Cntr=0.3,0.1

Type RM Length L Ch R = 1 ,82902   ,382,382,382
BEGIN DESCRIPTION:
STEWARTS CREEK 162.0
END DESCRIPTION:
XS GIS Cut Line= 3
      3824561.34      10138285.2      3824656.06      10136884.1
      3824727.04     10136114.26
#Sta/Elev= 30
  3595.7  284.35  3765.8  277.67  3880.5  276.34  3890.5  275.77  3910.1  271.48
  3915.1  271.75  3920.6  269.65  3930.6  269.19  3970.7  276.35  4020.8  278.45
  4241.3  278.26  4341.5  275.42  4391.6  275.45  4471.8  270.41  4742.4  260.18
  4862.7  259.48  4950.2  260.64  4962.9  259.96  4978.4  255.09  5013.1  257.37
  5033.2   260.7  5364.6     273  5485.1  281.23  5575.5  285.82  5614.6  286.41
  5625.7  288.19  5724.3  289.03  5729.3  291.03  5736.1  291.15  5773.1  290.46
#Mann= 3 , 0 , 0
  3595.7     .11       0  4950.2     .04       0  5033.2     .11       0
Bank Sta=4950.2,5033.2
XS Rating Curve= 0 ,0
Exp/Cntr=0.3,0.1

Type RM Length L Ch R = 1 ,82520   ,520,520,520
BEGIN DESCRIPTION:
Mapping XS 95122248
END DESCRIPTION:
XS GIS Cut Line= 3
       3824922.3      10138146.5      3825034.45     10136905.46
      3825016.06     10136167.29
#Sta/Elev= 30
  3753.9  282.09  3950.1  274.55  4010.4  275.26  4100.7  267.69  4221.2   266.2
  4442.1  267.13  4452.2  265.78    4488  265.93  4673.1  265.82  4703.2     270
  4719.3   269.3  4759.2  259.57  4764.2  260.51  4793.6  257.26  4883.9  258.84
    4914   257.3  4964.2  257.82  4980.8   255.5  4985.8  256.28  4989.8  254.19
    4999  254.19  4999.5  254.69  4999.7  257.44  5024.4  258.65  5078.3  261.81
    5258  276.59  5304.5   279.2  5580.3  284.85  5726.3  290.04  5738.4  290.24
#Mann= 9 ,-1 , 0
  3753.9     .17       0    4488     .11       0  4719.3     .15       0
  4883.9     .04       0  5024.4     .15       0  5078.3     .17       0
    5258     .11       0  5580.3     .17       0  5726.3     .11       0
#XS Ineff= 2 , 0
       0  4764.2  260.51               0
Permanent Ineff=
       F       F
Bank Sta=4883.9,5024.4
XS Rating Curve= 0 ,0
Exp/Cntr=0.3,0.1

Type RM Length L Ch R = 1 ,82000   ,500,500,500
BEGIN DESCRIPTION:
STEWARTS CREEK 161.0
END DESCRIPTION:
XS GIS Cut Line= 3
      3825245.22     10138167.32       3825518.6     10136855.41
      3825282.25     10136168.96
#Sta/Elev= 30
  3659.9   284.5  3737.8  282.37  3913.9  280.03  4350.7  270.58  4442.6  267.65
  4452.8  265.97  4687.8  265.74  4708.2  266.33  4725.1  269.24  4749.1  265.21
  4769.5  259.42  4780.3  255.13  4905.2  255.98  4943.1  255.83  4994.2  254.57
    4995  252.91  5004.3  252.91  5025.7  255.54    5045  254.93  5131.5   257.4
  5216.1  262.59  5320.7  267.18  5326.4  268.46  5351.9  268.78  5382.8  270.86
  5469.9  274.81  5539.3  280.42  5586.3  281.42  5670.9  286.14    5726   287.9
#Mann= 7 ,-1 , 0
  3659.9     .17       0  3913.9     .11       0  4905.2     .15       0
  4943.1     .04       0  5025.7     .15       0  5326.4     .17       0
  5382.8     .11       0
Bank Sta=4943.1,5025.7
XS Rating Curve= 0 ,0
Exp/Cntr=0.3,0.1

Type RM Length L Ch R = 1 ,81500   ,500,500,500
BEGIN DESCRIPTION:
STEWARTS CREEK 160.0
END DESCRIPTION:
XS GIS Cut Line= 3
      3826083.49      10137996.1      3825998.57     10136894.97
      3825899.25     10136158.14
#Sta/Elev= 30
  3895.6  286.46  4131.3  274.33  4239.9  270.93  4290.4  269.14  4321.9  269.48
    4342  267.81  4436.8  264.96  4536.6   260.8  4763.2  254.74  4816.3  251.76
  4873.5  253.11  4923.7  253.36  4933.7  252.15  4963.8  252.84  4983.9  252.29
  4994.7  249.85  5034.2  252.34  5104.8  254.68    5125  254.15  5155.3  255.17
  5165.4  256.62    5236  258.75  5330.4  265.34  5397.5  268.44  5414.9  270.37
  5419.9  269.78  5492.6  272.21  5498.4  273.43  5538.7  273.94  5743.5  280.73
#Mann= 7 ,-1 , 0
  3895.6     .17       0  4239.9     .11       0  4436.8     .17       0
  4536.6     .15       0  4763.2     .04       0  5104.8     .15       0
  5330.4     .11       0
Bank Sta=4763.2,5104.8
XS Rating Curve= 0 ,0
Exp/Cntr=0.3,0.1

Type RM Length L Ch R = 1 ,81000   ,500,500,500
BEGIN DESCRIPTION:
STEWARTS CREEK 159.0
END DESCRIPTION:
XS GIS Cut Line= 3
      3826794.12     10137768.04      3826463.67       10137053.
      3825969.46     10136149.42
#Sta/Elev= 30
  4212.3  283.97    4547  269.35  4561.5  267.48  4569.9  268.19    4716  255.87
  4770.8  253.88  4869.9  250.07    4892   251.4  4907.5  251.54    4925  249.61
  4981.9  251.15  4999.9     248  5009.8     248  5013.6  251.36  5093.4  253.85
  5167.9  257.93  5268.5  261.32  5396.5  264.64  5492.3  264.18  5542.5  262.73
  5565.4  262.38  5581.5  263.45  5587.2  265.58  5594.9  266.33  5652.7  268.91
  5810.1  271.41  5897.4   274.4  5925.4  276.68  5993.8  277.32  6029.9  279.86
#Mann= 6 ,-1 , 0
  4212.3     .17       0    4716     .15       0  4770.8     .04       0
  5093.4     .15       0  5268.5     .17       0  5542.5     .11       0
Bank Sta=4770.8,5093.4
XS Rating Curve= 0 ,0
Exp/Cntr=0.3,0.1

Type RM Length L Ch R = 1 ,80500   ,171,171,171
BEGIN DESCRIPTION:
STEWARTS CREEK 158.0
END DESCRIPTION:
XS GIS Cut Line= 3
      3827079.24     10137618.91      3826889.25     10136830.17
       3826666.9     10135728.28
#Sta/Elev= 30
  4188.7  284.44  4346.3  278.44  4419.1  274.77  4517.8  271.31  4596.5  265.67
  4638.5  265.02  4732.6   257.8  4885.9  252.95  4989.3  250.23    4992  248.33
  5141.9  252.66  5274.5  258.53  5287.5  262.76  5294.9  263.32  5325.5  259.97
  5383.9  262.56    5389  261.57  5417.3  266.64  5439.8  268.32  5458.2   268.1
  5485.5  264.62    5652  263.48  5693.7  264.47  5713.2  266.72  5739.4  265.86
  5744.5  267.17  5978.4  270.89    6009   274.5  6082.9  275.66  6124.1  275.79
#Mann= 6 ,-1 , 0
  4188.7     .11       0  4346.3     .17       0  4419.1     .11       0
  4885.9     .04       0  5141.9     .11       0  6082.9    .125       0
Bank Sta=4885.9,5141.9
XS Rating Curve= 0 ,0
Exp/Cntr=0.3,0.1

Type RM Length L Ch R = 1 ,80329   ,829,829,829
BEGIN DESCRIPTION:
STEWARTS CREEK 157.0
END DESCRIPTION:
XS GIS Cut Line= 3
      3827210.83     10137390.79      3827040.28     10136769.37
      3826817.24     10135594.25
#Sta/Elev= 30
  4355.6  281.26  4798.7  256.17  4811.6  257.31  4872.8  254.72  4957.2  253.57
 4982.84251.4585  4996.5  249.23  5023.8  248.03  5033.8  248.03    5042  251.44
  5094.2  254.26  5146.5  252.61  5151.6  253.72  5198.7  253.08  5203.8  254.41
    5251  254.38  5283.3  256.96  5405.4  260.31  5522.5  258.62    5627  258.92
  5632.1  260.52  5670.1  260.23  5684.3  261.86  5846.2  266.04  5893.4  264.42
  5914.3  266.88  5950.7  266.73  5955.8     268    6003  268.25  6196.1  274.53
#Mann= 3 , 0 , 0
  4355.6     .11       0 4982.84     .04       0    5042     .11       0
Bank Sta=4982.84,5042
XS Rating Curve= 0 ,0
Exp/Cntr=0.3,0.1

Type RM Length L Ch R = 1 ,79500   ,500,500,500
BEGIN DESCRIPTION:
STEWARTS CREEK 156.0
END DESCRIPTION:
XS GIS Cut Line= 3
      3827618.77     10137272.35      3827781.76     10136406.36
      3827745.98     10135658.11
#Sta/Elev= 30
  4118.8  283.07  4221.4  279.53  4338.6  275.67  4468.2   270.7  4547.5  266.66
  4630.7  261.38  4678.1  257.43  4683.2  257.85  4788.1  252.71  4845.7  251.54
  4893.1  249.91  4898.1  250.43  4950.6  247.76  4955.7  248.59  5040.2  246.57
  5075.4  247.66  5305.6  247.32  5345.7  248.69  5385.7  251.23  5445.8  255.13
  5455.8   256.7  5515.9  262.02  5555.9   262.4  5565.9  265.45  5575.9  267.05
    5596   268.8  5608.1  268.85    5636  271.89  5706.1   276.6  5749.1  278.35
#Mann= 5 ,-1 , 0
  4118.8     .17       0  4221.4     .11       0  4338.6     .17       0
  4845.7     .04       0  5385.7     .17       0
Bank Sta=4845.7,5385.7
XS Rating Curve= 0 ,0
Exp/Cntr=0.3,0.1

Type RM Length L Ch R = 1 ,79000   ,500,500,500
BEGIN DESCRIPTION:
STEWARTS CREEK 155.0
END DESCRIPTION:
XS GIS Cut Line= 3
      3828316.23     10137355.71      3828266.73     10136453.76
      3828355.64     10135645.54
#Sta/Elev= 30
  4096.7  277.59  4111.4  277.36  4121.4  276.22  4162.4  275.65  4248.3  271.13
  4391.8  264.52  4491.9  257.66  4520.2     257    4540  255.49  4591.2  253.58
  4602.1   252.8  4698.5  251.34  4722.3  251.59  4882.5  249.12  4902.5   248.1
  4952.6  248.19  5017.4  246.46  5042.9  247.64    5335  247.59    5421  251.53
  5465.5  253.42  5475.5  254.17    5487   256.4    5512  262.31    5517  261.65
  5535.9  262.95    5556  262.78  5585.5  264.27  5737.1  272.34  5813.1   272.8
#Mann= 9 ,-1 , 0
  4096.7     .11       0  4248.3     .17       0    4540     .11       0
  4591.2     .17       0  4698.5     .15       0  4722.3     .04       0
    5421     .11       0    5487     .17       0  5585.5    .125       0
Bank Sta=4722.3,5421
XS Rating Curve= 0 ,0
Exp/Cntr=0.3,0.1

Type RM Length L Ch R = 1 ,78500   ,500,500,500
BEGIN DESCRIPTION:
STEWARTS CREEK 154.0
END DESCRIPTION:
XS GIS Cut Line= 3
      3829000.52     10136908.24       3828740.5     10136349.03
      3828478.54     10135557.24
#Sta/Elev= 30
  4383.3  284.57  4450.4  284.29  4635.2  274.93  4745.6  268.12  4896.3  255.85
  4924.7  254.16  4947.6  251.67  4997.2  247.35  5156.4  247.62  5166.4  247.52
  5171.5  246.57  5214.6  247.69  5341.5  248.06  5346.7  247.51    5356  248.95
  5398.1  249.09  5450.8  251.52  5492.4  253.84  5523.7  256.08    5537   256.4
  5563.5  258.66  5626.9  261.53  5640.4  262.94  5695.6   265.5  5702.2  266.37
  5714.1  268.63  5722.1  271.43  5727.3  270.77  5735.2   271.7    5834  272.13
#Mann= 8 ,-1 , 0
  4383.3     .17       0  4635.2     .11       0  4745.6     .17       0
  4947.6     .04       0  5450.8     .11       0  5492.4     .17       0
  5523.7     .11       0  5702.2    .125       0
Bank Sta=4947.6,5450.8
XS Rating Curve= 0 ,0
Exp/Cntr=0.3,0.1

Type RM Length L Ch R = 1 ,78000   ,602,602,602
BEGIN DESCRIPTION:
STEWARTS CREEK 153.0
END DESCRIPTION:
XS GIS Cut Line= 3
      3829227.44     10136666.98      3829142.88      10136085.1
      3828571.74     10135492.54
#Sta/Elev= 30
    4412  276.68    4486  272.89  4539.2   270.4  4549.3  269.34  4585.9  268.12
  4700.9  261.87  4724.1  261.52  4731.2  260.51  4812.1  257.12  4842.4  253.17
  4864.4  251.74  4892.9  250.02  4917.2  247.27  4917.7  246.77  4928.7  246.77
  4929.5  247.58  4953.5  247.72    5367  247.52  5388.3  249.12  5395.3  248.74
  5451.9  251.92  5508.5  254.51  5522.6  256.03  5550.9  257.07  5621.7  262.57
  5661.3  264.36  5716.6  267.67  5770.1  270.48  5798.4  270.79    5823  272.74
#Mann= 7 ,-1 , 0
    4412     .17       0    4486     .11       0  4585.9     .17       0
  4864.4     .04       0  5451.9     .17       0  5661.3    .125       0
  5716.6     .11       0
Bank Sta=4864.4,5451.9
XS Rating Curve= 0 ,0
Exp/Cntr=0.3,0.1

Type RM Length L Ch R = 1 ,77398   ,117,117,117
BEGIN DESCRIPTION:
STEWARTS CREEK 152.0
END DESCRIPTION:
XS GIS Cut Line= 3
      3829772.57     10136123.08      3829580.89      10135798.1
      3828892.61     10135186.28
#Sta/Elev= 30
  4622.7  280.72  4679.2  280.09  4743.6   275.7  4774.9  271.78  4780.7  273.15
  4796.3  270.96  4802.1  272.43  4817.8   270.5  4823.6  271.39  4860.7  269.43
  4868.8  265.42  4876.3  259.85    4892  252.55  4897.8  251.24  4940.7  247.84
  4962.1  247.65  5573.9  247.68    5575   246.9  5602.3  247.79    5609  249.18
  5637.4  251.63  5722.7  257.73  5757.8  260.93  5779.6  263.87  5814.7  264.97
  5843.1  267.69  5849.8  267.06  5878.2  269.33  5885.8     269  5920.9  270.57
#Mann= 3 , 0 , 0
  4622.7     .11       0  4897.8     .04       0  5637.4     .17       0
Bank Sta=4897.8,5637.4
XS Rating Curve= 0 ,0
Exp/Cntr=0.3,0.1

Type RM Length L Ch R = 1 ,77281   ,71,71,71
BEGIN DESCRIPTION:
Mapping XS 2b0f7d15
END DESCRIPTION:
XS GIS Cut Line= 3
      3829798.88     10136101.16      3829664.05      10135716.3
      3829035.62     10135039.59
#Sta/Elev= 30
  4592.2  281.61  4719.4  278.35  4846.6  269.69  4877.9  258.76  4883.2  252.25
 4887.22251.2796  4934.3  249.34  5092.9  251.24  5192.1  258.94  5291.3  258.43
  5298.1  256.48  5305.5  258.23  5312.3  256.15  5319.6  257.79  5354.8  255.46
  5383.1  258.76  5489.2  255.19  5496.5  257.36  5520.1  255.03    5549  254.73
    5560  257.72    5581  254.69  5588.4  256.55  5595.2  254.12  5602.5  256.16
  5623.5  253.14  5630.9  255.24  5637.7  252.32  5779.4  265.12  5923.5  272.44
#Mann= 5 ,-1 , 0
  4592.2     .11       0 4887.22     .04       0  5092.9     .11       0
  5520.1     .15       0    5549     .17       0
#XS Ineff= 2 , 0
       0                  5177.9       0  258.67
Permanent Ineff=
       F       F
Bank Sta=4887.22,5092.9
XS Rating Curve= 0 ,0
Exp/Cntr=0.3,0.1

Type RM Length L Ch R = 1 ,77210   ,710,710,710
BEGIN DESCRIPTION:
STEWARTS CREEK 151.0
END DESCRIPTION:
XS GIS Cut Line= 3
      3829855.89     10136105.49      3829714.75     10135666.42
      3829075.85     10135005.28
#Sta/Elev= 30
  4538.8   281.7  4827.1   271.5  4869.1  263.51  4890.1  250.47  4944.4  247.19
  4965.6  244.95  5036.9  247.01  5057.6  246.33    5086  246.13  5121.8  252.77
  5176.3  247.72  5213.8  246.02  5234.9  249.19  5242.1  246.78  5249.1  249.35
  5256.3  247.16    5334  250.97  5341.2  248.62  5348.1  251.07  5362.3  246.71
  5425.8   250.6    5433   248.3    5440  250.91  5557.9  251.09  5609.7  253.26
  5616.9   250.6  5623.9  253.58  5631.1  251.33  5751.2  262.17  5919.4  270.74
#Mann= 7 ,-1 , 0
  4538.8     .11       0  4944.4     .04       0  5036.9     .11       0
  5057.6     .15       0    5086     .11       0  5176.3     .15       0
  5557.9     .17       0
#XS Ineff= 2 , 0
       0                  5121.8       0  252.77
Permanent Ineff=
       F       F
Bank Sta=4944.4,5036.9
XS Rating Curve= 0 ,0
Exp/Cntr=0.3,0.1

Type RM Length L Ch R = 1 ,76500   ,500,500,500
BEGIN DESCRIPTION:
STEWARTS CREEK 150.0
END DESCRIPTION:
XS GIS Cut Line= 3
      3830522.57     10135653.07      3829660.33     10135050.55
      3829100.93     10134962.41
#Sta/Elev= 30
  3948.1   267.5  4161.3  254.22  4240.1  253.37  4285.7  254.71  4356.1  256.73
  4419.3  255.55  4534.9  249.06  4617.7  245.99  4749.4     238  4807.8  238.74
  4850.6  237.16  4871.5  238.11    4916  237.35  4922.1  236.08  4951.8  236.56
  4957.9  235.39  4966.4  237.24  4972.7  236.22    4988  229.78  4999.2  229.78
  5003.8  232.41  5028.3  237.27  5035.5  237.33  5053.1  236.34  5090.8  237.23
  5255.6   247.3  5296.1  247.91  5336.6  253.82  5413.4   260.3  5566.3  268.74
#Mann= 7 ,-1 , 0
  3948.1     .11       0  4285.7     .17       0  4419.3     .11       0
  4617.7     .15       0  4966.4     .04       0  5028.3     .15       0
  5035.5     .17       0
Bank Sta=4966.4,5028.3
XS Rating Curve= 0 ,0
Exp/Cntr=0.3,0.1

Type RM Length L Ch R = 1 ,76000   ,500,500,500
BEGIN DESCRIPTION:
STEWARTS CREEK 149.0
END DESCRIPTION:
XS GIS Cut Line= 3
      3830880.22     10134823.21      3829936.92     10134658.31
      3829262.47     10134510.78
#Sta/Elev= 30
  4042.4  280.84  4087.2  278.17    4196  268.38  4248.6  265.86  4279.9  262.44
    4329  257.18  4440.7  249.05    4461  248.69  4493.5  245.64  4582.8  244.39
  4623.2  242.75  4714.8  240.24  4826.8  234.86  4846.8  235.23  4856.9   233.8
  4877.2  235.23  4959.2  234.73  4991.3  230.35  5002.6  230.35  5029.8  235.95
  5056.3  234.92  5104.9  236.51  5132.1  236.83  5154.3  239.07  5321.2  246.07
  5439.2  253.76  5459.7  254.29  5481.9  256.79  5618.6  266.19  5690.4  269.53
#Mann= 9 ,-1 , 0
  4042.4     .11       0  4248.6     .17       0  4279.9     .11       0
  4623.2     .17       0  4826.8     .15       0  4959.2     .04       0
  5029.8     .15       0  5104.9     .11       0  5321.2     .17       0
Bank Sta=4959.2,5029.8
XS Rating Curve= 0 ,0
Exp/Cntr=0.3,0.1

Type RM Length L Ch R = 1 ,75500   ,500,500,500
BEGIN DESCRIPTION:
STEWARTS CREEK 148.0
END DESCRIPTION:
XS GIS Cut Line= 3
      3830918.38     10134670.42      3830047.66     10134229.92
      3829283.11      10134396.1
#Sta/Elev= 30
  4024.2  279.91  4082.3  276.61    4099   274.7  4104.6  275.79  4126.8  274.23
  4143.5  271.38    4220  266.55  4349.8  255.91    4383  254.75  4388.6   253.4
  4440.9   250.6  4494.5  246.95  4500.1  247.95  4506.7  246.55  4561.3  243.49
  4703.4  237.74  4784.1  233.14  4798.1  233.92  4977.4  233.83  4984.6  229.12
    4996  229.12  4997.1  231.15  5002.5  231.15    5010  234.14  5029.3  233.37
  5076.3  234.82  5147.7  239.93  5276.1  248.22  5614.7  261.81  5782.4  268.52
#Mann= 9 ,-1 , 0
  4024.2     .11       0    4220     .17       0  4440.9     .11       0
  4703.4     .15       0  4977.4     .04       0    5010     .15       0
  5029.3     .17       0  5147.7     .11       0  5614.7     .17       0
Bank Sta=4977.4,5010
XS Rating Curve= 0 ,0
Exp/Cntr=0.3,0.1

Type RM Length L Ch R = 1 ,75000   ,500,500,500
BEGIN DESCRIPTION:
STEWARTS CREEK 147.0
END DESCRIPTION:
XS GIS Cut Line= 3
      3831106.81     10134370.11      3830304.69     10133848.88
      3829256.06     10133227.71
#Sta/Elev= 30
  4043.4  267.79    4122  266.71  4185.3  263.35  4303.2  259.97  4465.5  254.43
  4532.5  251.34  4547.7  251.93  4723.1  243.86  4858.7  236.61  4924.7   235.2
  4946.3  233.45  4973.4  231.76  4988.5  229.32  4989.4  228.08  5000.8  228.08
  5009.6  231.65  5019.4  233.44  5157.9  232.48  5379.4  233.59  5456.1  234.21
  5477.5  236.64    5499  237.18  5588.7  236.69    5616  238.18  5668.6  237.13
  5711.5  238.16  5937.8  248.14  6083.9  250.47    6189  256.05  6218.8   258.2
#Mann= 8 ,-1 , 0
  4043.4     .11       0  4303.2     .17       0  4465.5     .11       0
  4723.1     .15       0  4946.3     .04       0  5019.4     .15       0
  5379.4     .11       0    6189     .17       0
#XS Ineff= 2 ,-1
    5499    5624  237.18    5624  5717.3   238.2
Permanent Ineff=
       F       F
Bank Sta=4946.3,5019.4
XS Rating Curve= 0 ,0
Exp/Cntr=0.3,0.1

Type RM Length L Ch R = 1 ,74500   ,500,500,500
BEGIN DESCRIPTION:
STEWARTS CREEK 146.0
END DESCRIPTION:
XS GIS Cut Line= 3
      3831221.39     10133797.18      3830424.81     10133430.09
      3829473.59     10132805.58
#Sta/Elev= 30
  4122.9  264.03  4174.8  263.53  4226.3   260.8    4380  248.12  4490.2  241.15
  4765.4  233.01  4822.2   231.2    4960  232.44  4982.9  230.58  4988.4  229.11
  4989.6  227.34  5001.6  227.34  5010.8  230.64  5032.2  232.25  5092.1     231
  5098.2  229.32  5113.3  230.54  5119.3  229.75  5134.4  232.93  5230.4  237.63
  5294.1  238.64  5393.5  237.55  5459.9  239.82  5546.6  240.37  5574.4  241.83
  5682.8  242.51  5703.9  244.03  5734.1   243.7  5929.4  248.96  6137.9  256.33
#Mann= 5 ,-1 , 0
  4122.9     .11       0  4765.4     .15       0    4960     .04       0
  5032.2     .15       0  5230.4     .11       0
Bank Sta=4960,5032.2
XS Rating Curve= 0 ,0
Exp/Cntr=0.3,0.1

Type RM Length L Ch R = 1 ,74000   ,500,500,500
BEGIN DESCRIPTION:
STEWARTS CREEK 145.0
END DESCRIPTION:
XS GIS Cut Line= 3
      3831450.51     10133210.36      3830697.06     10133042.59
      3829652.35      10132509.2
#Sta/Elev= 30
  4228.1  263.83  4302.5  262.41  4387.7  257.87    4572  243.49  4712.7  235.67
  4835.3  232.85  4850.7  231.16    4866  229.98    4948  229.31  4978.7  231.22
    4989  230.03    4997  227.42  5031.8  230.94  5148.5  229.63  5164.7  226.66
  5176.8  226.66  5178.8   228.4  5209.5  231.71    5259  234.63  5298.4  237.02
  5342.9  237.39  5459.6  234.36  5509.2  236.05  5751.4  241.68  5809.6   243.7
  5831.8  245.72  5863.7  245.58  6092.9  253.36  6109.5  255.01    6173  256.31
#Mann= 6 ,-1 , 0
  4228.1     .11       0  4850.7     .15       0  4978.7     .04       0
  5031.8     .15       0    5259     .17       0  5509.2     .11       0
#XS Ineff= 2 , 0
       0  4756.2  235.26  5298.4       0  237.02
Permanent Ineff=
       F       F
Bank Sta=4978.7,5031.8
XS Rating Curve= 0 ,0
Exp/Cntr=0.3,0.1

Type RM Length L Ch R = 1 ,73500   ,500,500,500
BEGIN DESCRIPTION:
STEWARTS CREEK 144.0
END DESCRIPTION:
XS GIS Cut Line= 3
      3831481.78     10133057.59      3830826.63     10132594.67
      3829781.63     10132200.41
#Sta/Elev= 30
  4197.8  263.75  4240.3  263.47  4335.1  259.96  4427.4  254.25    4521  246.43
  4606.7  242.26  4650.3  237.59  4721.7  235.36    4793   230.9  4883.2  228.93
  4914.9  228.07    4974  229.74  4986.3  227.91  4992.7  224.66  5004.8  224.66
  5009.4  228.14  5019.5  229.83  5085.3   228.8  5104.8  227.41  5116.3  228.72
  5126.9  226.98  5285.3  229.35  5397.5  230.85  5543.8  233.34  5725.5  239.28
  5902.2  247.85  5917.9  247.75  5957.2  250.73  6102.9  256.53  6116.9  257.91
#Mann= 6 ,-1 , 0
  4197.8     .11       0  4883.2     .15       0    4974     .04       0
  5019.5     .15       0  5285.3     .17       0  5397.5     .11       0
Bank Sta=4974,5019.5
XS Rating Curve= 0 ,0
Exp/Cntr=0.3,0.1

Type RM Length L Ch R = 1 ,73000   ,500,500,500
BEGIN DESCRIPTION:
STEWARTS CREEK 143.0
END DESCRIPTION:
XS GIS Cut Line= 3
      3831551.25     10132930.89      3830938.18     10132132.14
      3830357.51     10131655.41
#Sta/Elev= 30
  3993.1   261.7  4073.7  259.62  4088.2  258.23    4109  258.82  4138.1  255.47
  4223.2  250.15  4266.8  245.95  4322.9  243.93  4358.4  241.15  4495.2   237.1
  4586.7  233.09  4651.1  231.72  4659.3   230.6    4681  230.74  4873.2  227.32
  4972.9  228.66  4987.6  223.82  4999.7  223.82  5008.2  227.74  5022.6  228.65
  5043.4  227.92  5065.1  225.77  5086.4  225.88  5202.5  231.45  5413.6  242.09
    5484  246.46  5576.5     254    5583  253.48  5675.6  256.94  5751.3  256.65
#Mann= 5 ,-1 , 0
  3993.1     .11       0    4681     .15       0  4972.9     .04       0
  5022.6     .15       0  5202.5     .11       0
Bank Sta=4972.9,5022.6
XS Rating Curve= 0 ,0
Exp/Cntr=0.3,0.1

Type RM Length L Ch R = 1 ,72500   ,500,500,500
BEGIN DESCRIPTION:
STEWARTS CREEK 142.0
END DESCRIPTION:
XS GIS Cut Line= 3
      3831685.78     10132826.71      3831243.49     10131771.34
      3830802.05     10131419.36
#Sta/Elev= 30
  3855.7  256.77  3926.9  255.38  3971.2  252.93  4013.4  252.41    4057  249.08
  4111.2  246.35  4154.6  242.49  4241.3   240.6  4338.9   236.4  4425.6  234.69
  4566.9  229.75  4716.9  225.95  4837.7  225.67  4979.9  227.25  4997.4  224.74
  4998.5   223.7  5010.7   223.7  5019.1  227.05  5060.7  226.99  5089.5  224.62
  5110.3  227.18  5182.4  233.05  5237.6  239.15  5310.5  246.35  5316.9  247.67
  5374.6  252.49  5380.9  252.27    5389  253.38  5502.7  259.98  5564.6  260.03
#Mann= 5 ,-1 , 0
  3855.7     .11       0  4716.9     .15       0  4979.9     .04       0
  5019.1     .15       0  5237.6     .11       0
Bank Sta=4979.9,5019.1
XS Rating Curve= 0 ,0
Exp/Cntr=0.3,0.1

Type RM Length L Ch R = 1 ,72000   ,500,500,500
BEGIN DESCRIPTION:
STEWARTS CREEK 141.0
END DESCRIPTION:
XS GIS Cut Line= 3
      3833152.81     10132535.91      3831466.72     10131414.79
      3830812.25     10131390.94
#Sta/Elev= 30
  2975.2  247.62  3335.8  244.61  3912.9  233.97  3985.1  235.13  4021.2  233.18
  4142.7  233.15  4258.7  231.31  4330.5  231.91  4374.2  232.46  4396.9  228.74
  4410.2   224.4    4424  229.46  4446.2  232.61  4460.1  231.31  4590.5  231.33
  4640.4   231.4  4799.8  223.93  4835.8  224.25  4836.4  223.17  4886.9  225.61
  4986.6  224.95  4995.2  223.73  5018.9  226.12  5058.9  225.05    5159  231.14
  5251.2  238.07  5469.2  249.83  5549.2  256.07  5619.3  259.44  5654.9  259.41
#Mann= 7 ,-1 , 0
  2975.2     .11       0  4142.7     .15       0  4330.5     .17       0
  4590.5     .11       0  4640.4     .04       0    5159     .15       0
  5251.2     .11       0
#XS Ineff= 2 , 0
       0  4446.2  232.61               0
Permanent Ineff=
       F       F
Bank Sta=4640.4,5159
XS Rating Curve= 0 ,0
Exp/Cntr=0.3,0.1

Type RM Length L Ch R = 1 ,71500   ,500,500,500
BEGIN DESCRIPTION:
STEWARTS CREEK 140.0
END DESCRIPTION:
XS GIS Cut Line= 3
      3833769.99     10131147.86      3831499.58     10131065.53
      3830711.93     10131116.55
#Sta/Elev= 30
  2728.1  249.94  3150.5  244.52  3332.5  240.68  3527.9   233.3  3574.2  231.98
    3831  227.49    3871  225.12    3951  225.89    3961  224.23  4031.1  228.88
  4071.1  225.83  4090.4  227.37  4161.7  228.17  4191.2  223.18  4221.2  227.91
  4261.2  226.76  4350.9  228.58  4531.4  230.89  4611.5  229.47  4845.5  222.68
  4881.6  225.11  5003.4  223.31  5041.8  226.18  5081.9   224.4    5152  225.33
  5302.4  229.95  5374.6  232.49  5542.9  241.48  5703.2  254.67  5789.3  256.93
#Mann= 8 ,-1 , 0
  2728.1     .11       0  3527.9     .17       0  3574.2     .11       0
  4090.4     .17       0  4350.9     .15       0  4611.5     .04       0
  5302.4     .11       0  5374.6     .11       0
#XS Ineff= 2 , 0
       0  4531.4  230.89               0
Permanent Ineff=
       F       F
Bank Sta=4611.5,5302.4
XS Rating Curve= 0 ,0
Exp/Cntr=0.3,0.1

Type RM Length L Ch R = 1 ,71000   ,500,500,500
BEGIN DESCRIPTION:
STEWARTS CREEK 139.0
END DESCRIPTION:
XS GIS Cut Line= 3
      3833514.73     10130897.86      3831553.53     10130748.26
      3831036.48     10130502.91
#Sta/Elev= 30
  3033.1  249.85  3270.7  247.31  3471.2  243.25  3585.9  239.08  3972.3  223.27
  4006.5  223.66  4042.9  228.21    4073  224.07    4083  224.89  4103.1   223.1
  4108.3  225.73  4143.2  225.94  4173.3  228.73  4230.7   227.7  4333.7  227.84
    4428  230.04  4625.4  229.02  4668.5  227.96  4694.8  226.61    4775  222.85
  4865.3  223.17  4887.6  221.26  4975.6  223.22  5008.5  222.15  5093.8  226.88
  5190.3  234.65  5332.2   240.8  5349.4  240.22  5504.4  251.92  5572.3  251.57
#Mann= 9 ,-1 , 0
  3033.1     .11       0  3585.9     .17       0  4006.5     .11       0
  4230.7     .15       0    4428     .11       0  4625.4     .17       0
  4668.5     .15       0  4694.8     .04       0  5093.8     .11       0
Levee=-1,4414,230.36,0,,,,
Bank Sta=4694.8,5093.8
XS Rating Curve= 0 ,0
Exp/Cntr=0.3,0.1

Type RM Length L Ch R = 1 ,70500   ,500,500,500
BEGIN DESCRIPTION:
STEWARTS CREEK 138.0
END DESCRIPTION:
XS GIS Cut Line= 3
       3833462.7     10130806.72      3831788.37      10130510.1
      3831071.98     10130442.21
#Sta/Elev= 30
  3299.6  248.69  3527.7  246.96  3836.4  238.62  3969.5  232.21  4068.1  227.74
  4186.2  222.69  4208.4  223.64  4222.1  225.42  4228.7  228.03  4269.3   222.8
  4309.9  224.87  4335.3   221.3  4340.4  223.51  4352.2  224.61  4366.8  225.04
  4451.7   226.9  4551.2  226.86  4650.8   228.1  4750.3  228.63    4899  227.04
  4980.2  222.59  4991.5  220.21  5030.7   222.4  5241.6  222.56  5419.5  234.69
  5443.6  236.32  5492.7     240    5563  248.66  5633.3  252.31  5719.6  250.63
#Mann= 15 ,-1 , 0
  3299.6     .11       0  3836.4     .17       0  3969.5     .11       0
  4068.1     .17       0  4186.2     .11       0  4352.2     .17       0
  4366.8     .11       0  4451.7     .15       0  4551.2     .11       0
  4650.8     .15       0  4750.3     .17       0  4980.2     .04       0
  5030.7     .17       0  5419.5     .15       0  5443.6     .11       0
#XS Ineff= 2 , 0
       0  4777.1  229.09               0
Permanent Ineff=
       F       F
Bank Sta=4980.2,5030.7
XS Rating Curve= 0 ,0
Exp/Cntr=0.3,0.1

Type RM Length L Ch R = 1 ,70000   ,500,500,500
BEGIN DESCRIPTION:
STEWARTS CREEK 137.0
END DESCRIPTION:
XS GIS Cut Line= 3
      3833454.04     10130754.65      3831838.22      10130178.7
      3831435.79     10130003.78
#Sta/Elev= 30
  3284.6  248.65  3488.2   247.4  3760.3  241.98    3909  236.96  3934.5  234.73
  4144.9  225.58  4161.7  223.27  4182.9  223.96  4214.8  227.85  4237.4  225.49
  4257.3  221.25    4263  222.35  4342.2  224.05  4363.4  219.99  4385.8  224.59
  4473.3  222.11    4512  223.95    4573  224.55  4582.9  224.44  4699.3  224.46
  4796.4   222.8  4863.3  220.65  4968.5  220.65  4991.3  218.67  5053.1  222.97
  5181.3  231.71  5251.2  234.84  5379.7  244.97  5409.4  246.02  5438.8  247.69
#Mann= 9 ,-1 , 0
  3284.6     .11       0    4263     .17       0  4385.8     .15       0
    4573     .11       0  4582.9     .15       0  4699.3     .17       0
  4796.4     .04       0  5053.1     .17       0  5409.4     .11       0
#XS Ineff= 2 , 0
       0  4214.8  227.85               0
Permanent Ineff=
       F       F
Bank Sta=4796.4,5053.1
XS Rating Curve= 0 ,0
Exp/Cntr=0.3,0.1

Type RM Length L Ch R = 1 ,69500   ,500,500,500
BEGIN DESCRIPTION:
STEWARTS CREEK 136.0
END DESCRIPTION:
XS GIS Cut Line= 3
      3833336.79     10130637.44      3832207.95     10130097.79
      3831583.37     10129830.17
#Sta/Elev= 30
  3748.8  247.12  4149.2  241.58  4313.4  236.06  4494.8  226.87    4512  224.43
  4534.6  224.85  4556.7  227.53  4578.9  225.95  4585.5  223.12  4601.1  221.87
  4633.1  222.46  4676.3  221.31  4698.9  223.33  4704.5  223.11  4711.9  219.97
  4721.6  220.03  4734.1  223.68  4749.8   223.9  4811.7  222.04  4966.9  221.12
  5002.2  219.03    5011  221.16  5081.1  221.21  5113.6  218.36  5141.5  220.73
  5204.4   220.5  5275.6  223.25  5438.4  230.25  5542.2  237.55  5679.5  245.93
#Mann= 6 ,-1 , 0
  3748.8     .11       0  4633.1     .15       0  4966.9     .04       0
    5011     .15       0  5275.6     .17       0  5542.2     .11       0
#XS Ineff= 2 , 0
       0  4556.7  227.53               0
Permanent Ineff=
       F       F
Bank Sta=4966.9,5011
XS Rating Curve= 0 ,0
Exp/Cntr=0.3,0.1

Type RM Length L Ch R = 1 ,69000   ,500,500,500
BEGIN DESCRIPTION:
STEWARTS CREEK 135.0
END DESCRIPTION:
XS GIS Cut Line= 3
       3833371.5       10130581.      3832383.98     10129750.38
      3831596.32     10129786.75
#Sta/Elev= 30
  3709.6  245.95  4045.5  241.11  4273.1  241.41  4351.2  238.37  4529.6  228.47
  4599.6  223.53  4642.1  226.67  4655.6  225.32  4677.6   220.8  4691.9  221.87
  4790.8   220.8  4868.8  221.92  4932.6  220.66  4946.9   222.1  4975.5  220.98
    4982  219.58  4982.2  216.86  4982.7  216.36  4996.8  216.36  5006.1  219.37
  5016.2  220.68  5066.2   220.7  5116.3  222.76  5127.4  224.22  5159.8  224.74
  5256.4  228.52  5496.7  234.82  5606.8  236.36  5682.9  240.09  5788.5  245.44
#Mann= 6 ,-1 , 0
  3709.6     .11       0  4529.6     .15       0  4975.5     .04       0
  5016.2     .15       0  5159.8     .17       0  5682.9     .11       0
#XS Ineff= 2 , 0
       0  4642.1  226.67               0
Permanent Ineff=
       F       F
Bank Sta=4975.5,5016.2
XS Rating Curve= 0 ,0
Exp/Cntr=0.3,0.1

Type RM Length L Ch R = 1 ,68500   ,500,500,500
BEGIN DESCRIPTION:
STEWARTS CREEK 134.0
END DESCRIPTION:
XS GIS Cut Line= 3
      3833697.02     10130485.51      3832511.42     10129443.25
      3831987.93     10128884.99
#Sta/Elev= 30
  3421.4  243.92  3738.2  239.29  3912.6  236.22  4217.9  232.58  4294.2  229.75
  4472.2  222.12  4536.7  221.69  4557.6  220.18  4614.5     223  4670.4  223.56
  4685.2  223.18  4720.8  226.17  4770.1   222.1  4798.6  226.99  4812.8  227.07
  4913.1   221.9    4976  220.57  4982.7  219.43  4989.9  216.07    5004  216.07
  5004.9  218.19    5018  220.95  5138.7  219.16    5188  220.76    5273  218.36
  5386.3  219.94  5438.9  224.37  5690.1  242.11  5725.8  244.22  5765.3   244.1
#Mann= 9 ,-1 , 0
  3421.4     .11       0  3738.2     .17       0  3912.6     .11       0
  4294.2     .17       0  4670.4     .11       0  4913.1     .15       0
    4976     .04       0    5018     .15       0  5438.9     .11       0
Bank Sta=4976,5018
XS Rating Curve= 0 ,0
Exp/Cntr=0.3,0.1

Type RM Length L Ch R = 1 ,68000   ,531,531,531
BEGIN DESCRIPTION:
STEWARTS CREEK 133.0
END DESCRIPTION:
XS GIS Cut Line= 3
      3834005.26     10129443.88      3832538.19     10129042.83
      3832013.06     10128823.22
#Sta/Elev= 30
  3479.1  248.26  3569.7  246.22    3616  243.49  3939.4  229.45  4040.7  225.95
  4141.9  222.52  4228.6   219.4  4363.5   218.5  4421.9  219.62  4456.4  221.64
  4627.1   224.1  4644.6  221.66    4679  221.28  4718.8  224.49  4751.5  219.13
  4772.3  220.62  4856.9  218.94  4912.1  218.76  4958.9   220.1  4979.6  219.07
  4990.2  215.37    5005  215.37  5011.2  218.56  5017.1  218.96  5040.9  217.82
  5108.8  217.75  5283.4  228.71  5483.4  242.15  5560.2  244.61  5569.2  243.96
#Mann= 10 ,-1 , 0
  3479.1     .17       0    3616     .11       0  3939.4     .17       0
  4040.7     .11       0  4141.9     .17       0  4363.5     .11       0
  4856.9     .15       0  4979.6     .04       0  5017.1     .15       0
  5283.4     .11       0
Bank Sta=4979.6,5017.1
XS Rating Curve= 0 ,0
Exp/Cntr=0.3,0.1

Type RM Length L Ch R = 1 ,67469   ,469,469,469
BEGIN DESCRIPTION:
STEWARTS CREEK 132.0
END DESCRIPTION:
XS GIS Cut Line= 3
      3833922.74     10129174.77       3832583.9     10128678.67
      3832001.46     10128757.91
#Sta/Elev= 30
  3572.2  247.82  3716.9  242.83  3846.3  233.63  3913.6   229.1    4146  220.03
  4256.9  218.02  4465.2  217.06  4583.7  216.87  4666.3  217.53  4675.9  220.32
  4697.2  222.73  4729.2  215.81  4782.5  218.35  4846.5  217.99  4899.8  219.46
  4979.2  218.57  4987.8  214.17  5002.6  214.17  5006.1  215.74  5016.2  216.57
  5036.4  216.01 5050.66218.5363  5053.2  218.76  5058.3  216.03  5076.7  218.47
    5107  217.05  5175.6  218.23  5275.5  223.16  5470.3  237.82  5587.8  243.19
#Mann= 7 ,-1 , 0
  3572.2     .11       0  3846.3     .17       0  4465.2     .11       0
  4583.7     .15       0  4979.2     .04       0 5050.66     .15       0
  5175.6     .11       0
Bank Sta=4979.2,5050.66
XS Rating Curve= 0 ,0
Exp/Cntr=0.3,0.1

Type RM Length L Ch R = 1 ,67000   ,500,500,500
BEGIN DESCRIPTION:
STEWARTS CREEK 131.0
END DESCRIPTION:
XS GIS Cut Line= 3
      3833914.06      10129027.2      3832468.61      10128277.5
      3831856.77     10128241.61
#Sta/Elev= 30
  3371.7  246.28  3589.2  232.79  3691.8  227.68  3782.7  223.57  3937.6  222.93
  3987.5  224.15  4219.6  221.08  4224.7  220.16  4350.1   216.9  4457.3  216.76
  4493.9     222  4516.5  219.21  4523.7  216.69    4539  215.76  4551.4  217.97
  4617.8  215.34  4967.1  217.27    4977  215.15  4982.2  211.82    4997  211.82
  4997.5  212.32  4997.6  215.14  5010.8  216.95  5196.1  215.82  5291.3  220.15
  5347.4  224.23  5431.5  231.28  5471.6  236.18  5521.7   238.9  5612.9  241.48
#Mann= 8 ,-1 , 0
  3371.7     .11       0  3691.8     .17       0  4224.7     .11       0
  4350.1     .15       0  4967.1     .04       0  5010.8     .15       0
  5196.1     .17       0  5347.4     .11       0
Bank Sta=4967.1,5010.8
XS Rating Curve= 0 ,0
Exp/Cntr=0.3,0.1

Type RM Length L Ch R = 1 ,66500   ,500,500,500
BEGIN DESCRIPTION:
STEWARTS CREEK 130.0
END DESCRIPTION:
XS GIS Cut Line= 3
      3833979.14     10128896.98       3832701.8     10128117.85
      3832264.78     10127282.46
#Sta/Elev= 30
  3503.8   243.5  3734.8  230.45  3884.8  225.41  4199.6  222.17  4399.2  217.16
  4447.4  217.63  4462.8  215.79  4499.6   216.4  4512.7  218.68  4542.2  216.67
  4594.5  218.42  4652.6  215.65  4695.2  221.26  4737.8  215.22  4754.3  216.65
  4970.2  216.91  4979.8  214.67  4985.6  216.53    4992  210.78  5006.8  210.78
  5007.7   212.3  5021.9  215.01    5044  216.73  5446.5  215.04  5577.3  220.71
  5639.5  224.67  5758.8  237.53  5841.3  243.24  5926.4  249.12  5942.8  248.17
#Mann= 9 ,-1 , 0
  3503.8     .11       0  3884.8     .17       0  4399.2     .11       0
  4754.3     .15       0  4985.6     .04       0    5044     .15       0
  5577.3     .17       0  5758.8     .11       0  5841.3     .17       0
Bank Sta=4985.6,5044
XS Rating Curve= 0 ,0
Exp/Cntr=0.3,0.1

Type RM Length L Ch R = 1 ,66000   ,500,500,500
BEGIN DESCRIPTION:
STEWARTS CREEK 129.0
END DESCRIPTION:
XS GIS Cut Line= 3
      3833783.83     10128215.57      3832923.92      10127995.2
       3832326.1      10127235.4
#Sta/Elev= 30
  4112.3  238.48  4116.9  238.39  4234.2  234.99  4370.8  227.33  4463.4   223.5
  4521.1  221.44  4636.7  221.65  4779.2  221.09  4820.4  219.86  4861.7  215.14
  4876.4  215.41    4902  218.99  4917.2  220.65  4944.3  214.62    4965  214.28
  4978.1  210.56  4993.2  210.56  4998.2  213.79  5006.7  214.54  5035.6  215.84
  5078.9  213.45  5099.7  216.53  5157.5  216.85  5178.3   215.4  5370.8  213.27
  5528.4  218.56  5718.7  226.93  5832.4   237.4  5890.4   241.9  5966.8  250.54
#Mann= 10 ,-1 , 0
  4112.3     .11       0  4116.9     .17       0  4370.8     .11       0
  4463.4     .17       0  4636.7     .11       0    4902     .15       0
    4965     .04       0  5006.7     .15       0  5528.4     .17       0
  5832.4     .11       0
Bank Sta=4965,5006.7
XS Rating Curve= 0 ,0
Exp/Cntr=0.3,0.1

Type RM Length L Ch R = 1 ,65500   ,500,500,500
BEGIN DESCRIPTION:
STEWARTS CREEK 128.0
END DESCRIPTION:
XS GIS Cut Line= 3
       3833796.9     10128185.21      3832912.89     10127548.91
      3832364.98     10127195.86
#Sta/Elev= 30
  3910.8  237.45  3921.1  237.77  4008.1  236.64  4153.4  232.21  4171.2  231.29
    4416  221.16  4481.2  219.87  4614.7  218.73  4736.1   212.8  4801.2  219.78
  4815.3  218.67  4858.4  212.32  4895.3  215.38  4937.4   211.5  4966.9  215.09
  4987.7   213.3    4995  209.28  5010.2  209.28  5023.8  214.93  5053.6   210.1
  5075.3  209.96  5089.3  210.71  5096.4  215.93  5152.3  217.43  5199.8  218.63
  5301.3  221.97  5386.7  226.02  5545.3  239.08  5631.7  246.82  5651.8  251.57
#Mann= 15 ,-1 , 0
  3910.8     .11       0  3921.1     .17       0  4008.1     .11       0
  4153.4     .17       0  4171.2     .11       0    4416     .17       0
  4481.2     .11       0  4614.7     .17       0  4815.3     .15       0
  4966.9     .04       0  5023.8     .15       0  5152.3     .17       0
  5199.8     .15       0  5301.3     .17       0  5545.3     .11       0
Bank Sta=4966.9,5023.8
XS Rating Curve= 0 ,0
Exp/Cntr=0.3,0.1

Type RM Length L Ch R = 1 ,65000   ,500,500,500
BEGIN DESCRIPTION:
STEWARTS CREEK 127.0
END DESCRIPTION:
XS GIS Cut Line= 3
      3833814.21     10128159.11      3833079.69     10127203.61
      3832577.25     10126930.85
#Sta/Elev= 30
  3794.8  236.91  3819.9  236.43    3844  235.83  4035.3  231.71  4289.9  221.39
  4439.4  222.71  4566.6  217.63  4614.8  216.46  4661.5  214.12  4775.7  214.26
  4846.3  211.92  4860.8  212.25  4875.4  214.26  4881.7  217.01  4910.7  220.21
  4925.2  218.78  4931.5  215.58    4946  212.23  4995.9  212.69  4998.4  210.17
  5004.2  208.56  5019.4  208.56  5024.8  212.07  5033.6  212.64  5039.3  214.82
  5115.4  215.08  5253.1  224.04  5350.1  230.83  5400.3  232.13  5571.7  242.28
#Mann= 9 ,-1 , 0
  3794.8     .11       0  3819.9     .17       0    3844     .11       0
  4035.3     .17       0  4566.6     .11       0  4614.8     .15       0
  4995.9     .04       0  5033.6     .15       0  5253.1     .17       0
#XS Ineff= 2 , 0
       0  4902.5  220.18               0
Permanent Ineff=
       F       F
Bank Sta=4995.9,5033.6
XS Rating Curve= 0 ,0
Exp/Cntr=0.3,0.1

Type RM Length L Ch R = 1 ,64500   ,500,500,500
BEGIN DESCRIPTION:
STEWARTS CREEK 126.0
END DESCRIPTION:
XS GIS Cut Line= 3
      3834144.09     10127525.46      3833357.43     10126853.02
      3832638.07     10126748.56
#Sta/Elev= 30
  3965.1  236.27  4029.5  236.81  4035.7  236.58  4168.1  229.99  4256.4  225.21
  4355.2  222.31  4433.8  221.82  4490.2  219.38  4574.1  220.12  4686.6  219.07
  4816.2  211.86  4866.7  210.84    4959  213.56  4977.5212.1695  4986.4  210.24
    4990  206.92  5005.3  206.92  5009.7  210.18  5019.8  212.02  5070.3  211.02
  5110.7  212.75  5130.9  219.15    5141  220.63  5161.2  218.58  5171.4  214.33
  5199.1  213.34  5221.5  213.83  5467.7  222.15  5569.8  228.56  5726.9  237.66
#Mann= 11 ,-1 , 0
  3965.1     .11       0  4029.5     .15       0  4035.7     .11       0
  4168.1     .17       0  4574.1     .11       0  4686.6     .15       0
  4977.5     .04       0  5019.8     .15       0  5199.1     .11       0
  5221.5     .15       0  5569.8     .11       0
#XS Ineff= 2 , 0
       0                    5141       0  220.63
Permanent Ineff=
       F       F
Bank Sta=4977.5,5019.8
XS Rating Curve= 0 ,0
Exp/Cntr=0.3,0.1

Type RM Length L Ch R = 1 ,64000   ,600,600,600
BEGIN DESCRIPTION:
STEWARTS CREEK 125.0
END DESCRIPTION:
XS GIS Cut Line= 3
      3834387.18     10127121.84      3833518.15     10126458.13
      3832672.82     10126522.86
#Sta/Elev= 30
  3906.5  233.34    3943   233.4    3956  231.27  3970.2  232.29  4184.2  222.17
  4370.9   218.4  4534.8  218.23  4691.2  213.42  4770.2  210.31    4791  208.25
  4805.5  210.97  4834.6  211.73  4849.1  210.66    4976  212.37  4984.2  209.61
  4989.3  205.75  5004.7  205.75  5020.4  211.52  5030.4   212.5  5045.3   212.7
  5140.7  217.65  5180.8  216.48  5230.5  221.85    5251  222.07  5281.1  219.68
  5301.2  221.81  5401.5  223.81  5451.6  227.39  5496.8  228.77  5847.8  236.03
#Mann= 5 ,-1 , 0
  3906.5     .11       0  4370.9     .15       0    4976     .04       0
  5030.4     .15       0  5045.3     .11       0
#XS Ineff= 2 , 0
       0                  5140.7       0  217.65
Permanent Ineff=
       F       F
Bank Sta=4976,5030.4
XS Rating Curve= 0 ,0
Exp/Cntr=0.3,0.1

Type RM Length L Ch R = 1 ,63400   ,862,862,862
BEGIN DESCRIPTION:
STEWARTS CREEK 124.0
END DESCRIPTION:
XS GIS Cut Line= 3
      3834422.72     10126866.57      3833780.33     10126057.73
      3832677.12     10126278.07
#Sta/Elev= 30
  3967.1  229.42  3996.2  229.02  4159.6   220.6  4258.9  217.52  4308.5  216.44
  4337.4  217.87  4415.9  218.27  4616.6  213.24  4672.2  211.03  4771.6  209.89
  4778.6  208.84  4795.6  209.68  4825.4  211.14  4864.5  209.83  4970.2  211.01
  4978.2  210.03  4990.3  204.89  5005.7  204.89  5022.9   210.6  5033.1  211.05
  5265.2  212.04  5401.4  217.41  5420.6  218.16  5448.6  223.04  5461.4  222.88
  5481.8   219.8  5512.4  222.33  5573.6  223.37  5703.7   223.1    6125  229.18
#Mann= 8 ,-1 , 0
  3967.1     .11       0  4616.6     .15       0  4795.6     .11       0
  4825.4     .15       0  4970.2     .04       0  5033.1     .15       0
  5265.2     .17       0  5401.4     .11       0
Bank Sta=4970.2,5033.1
XS Rating Curve= 0 ,0
Exp/Cntr=0.3,0.1

Type RM Length L Ch R = 1 ,62538   ,538,538,538
BEGIN DESCRIPTION:
STEWARTS CREEK 123.0
END DESCRIPTION:
XS GIS Cut Line= 3
      3834391.48     10126049.74      3834191.87     10125692.41
      3832993.92      10124782.4
#Sta/Elev= 30
  4590.7  233.65  4645.1  226.19  4672.5  212.34  4731.9  208.63  4808.5   208.7
  4975.2  209.56  4980.9  207.22  4982.3  203.57  4997.8  203.57    4999  206.48
  5017.6  209.27  5154.4  210.03  5250.8  214.28  5360.3  218.59  5478.6  217.99
  5717.2  211.66  5720.3  211.81  5824.1  212.57  5853.2  224.22    5874  223.45
  5903.1  211.47  5938.4  209.25    5962  210.65  6017.4  214.39  6052.8  226.67
  6082.5   228.3  6202.9  228.45  6431.3  228.81  6452.1  233.89  6504.4  236.37
#Mann= 11 ,-1 , 0
  4590.7     .11       0  4808.5     .15       0  4975.2     .04       0
  5017.6     .15       0  5250.8     .17       0  5478.6     .15       0
  5717.2     .17       0  5720.3     .15       0    5962     .11       0
  6082.5    .125       0  6202.9     .15       0
#XS Ineff= 2 , 0
       0                  5439.3       0  218.94
Permanent Ineff=
       F       F
Bank Sta=4975.2,5017.6
XS Rating Curve= 0 ,0
Exp/Cntr=0.3,0.1

Type RM Length L Ch R = 1 ,62000   ,538,538,538
BEGIN DESCRIPTION:
STEWARTS CREEK 122.0
END DESCRIPTION:
XS GIS Cut Line= 3
      3834408.85     10126038.51       3834525.5     10125556.52
      3833582.66     10124677.55
#Sta/Elev= 30
  4504.1   231.7  4542.6  226.69  4607.8  222.13  4644.5  210.52  4649.6  211.77
  4717.5  208.34    4913   208.3  4947.6  205.82  4974.7  208.93  4984.3  206.66
  4987.3  204.12  5002.8  204.12  5016.3  208.06  5030.5  208.88  5267.7  211.37
  5320.7  210.98    5434  214.67  5497.9  213.77  5631.9  209.39  5737.9   210.3
  5752.1   209.4  5766.2  205.35  5787.7  210.07  5808.7  208.36  5841.5  210.43
  5936.2  209.47  6007.1  212.04  6212.3  222.17  6254.6  228.66    6289  229.64
#Mann= 6 ,-1 , 0
  4504.1     .11       0  4974.7     .04       0  5030.5     .15       0
  5267.7     .17       0  5497.9     .15       0  5841.5     .11       0
#XS Ineff= 2 ,-1
  5235.7  5355.8  212.03    5434  6070.6  214.67
Permanent Ineff=
       F       F
Bank Sta=4974.7,5030.5
XS Rating Curve= 0 ,0
Exp/Cntr=0.3,0.1

Type RM Length L Ch R = 1 ,61462   ,527,527,527
BEGIN DESCRIPTION:
STEWARTS CREEK 121.0
END DESCRIPTION:
XS GIS Cut Line= 3
      3835334.19     10126048.89      3834730.81     10125393.56
      3833761.67      10124678.3
#Sta/Elev= 30
  4109.2   232.2  4189.8  230.71  4347.6  220.22    4591   209.8  4642.4  207.96
  4778.7  207.65  4862.4  207.77  4904.9   203.5  4975.8  207.48    4982  202.29
  4997.6  202.29    5000  205.27  5011.2  207.45  5082.2  207.88    5150   211.7
  5276.5   216.4  5453.9   211.2  5518.1  211.13  5653.4  208.36  5698.3  209.63
  5704.5  208.19  5712.1  202.96  5733.7  208.36  5748.4   209.4  5884.1   209.3
  6019.8  213.18    6120  217.61  6155.5  223.32  6161.7  227.26  6204.5  229.45
#Mann= 10 ,-1 , 0
  4109.2     .11       0  4347.6     .17       0    4591     .15       0
  4642.4     .11       0  4778.7     .15       0  4975.8     .04       0
  5011.2     .15       0    5150     .17       0  5518.1     .15       0
  5653.4     .11       0
#XS Ineff= 2 , 0
       0                  5247.2       0  216.33
Permanent Ineff=
       F       F
Bank Sta=4975.8,5011.2
XS Rating Curve= 0 ,0
Exp/Cntr=0.3,0.1

Type RM Length L Ch R = 1 ,60935   ,672,672,672
BEGIN DESCRIPTION:
STEWARTS CREEK 120.0
END DESCRIPTION:
XS GIS Cut Line= 3
      3835365.47     10126028.12      3835121.89     10125143.13
       3833952.1       10124682.
#Sta/Elev= 30
  4082.1  230.88  4172.4  228.19  4265.7  221.76  4405.8  215.86  4556.1  210.23
  4680.6  210.88  4701.3  210.45  4722.1   207.7  4742.8  210.26  4917.5  206.66
    4971  206.17  4981.4  203.59  5025.8  207.02  5320.3  207.47  5350.1  206.15
  5507.1  208.07    5531  204.62  5534.2  202.25  5550.3  202.25  5552.5  204.25
  5566.6     208  5674.9  206.94  5921.6  209.75  6132.4  214.36  6162.2  216.46
  6167.5  219.71  6186.5   220.2  6191.9  223.99  6256.7  227.35  6257.4  227.37
#Mann= 8 ,-1 , 0
  4082.1     .11       0  4405.8     .17       0  4917.5     .04       0
  5025.8     .11       0  5507.1     .12       0  5566.6     .11       0
  5921.6     .15       0  6256.7     .11       0
#XS Ineff= 2 , 0
       0  4680.6  210.88               0
Permanent Ineff=
       F       F
Bank Sta=4917.5,5025.8
XS Rating Curve= 0 ,0
Exp/Cntr=0.3,0.1
