HEC-RAS study WFSJ Main.prj: WFSJ Main Base Level Engineering

--- WFSJ Main.g01 (geometry) --- (continued)

Type RM Length L Ch R = 1 ,232000  ,1000,1000,1000
BEGIN DESCRIPTION:
WFSJ Main 231.0
END DESCRIPTION:
XS GIS Cut Line= 3
      3841779.09     10090126.27      3840009.62     10085810.43
      3838622.84     10079641.89
#Sta/Elev= 30
   335.5  138.54    1406  117.43  1443.5  106.67  1512.8  120.58  1774.3  113.02
  2729.7  119.57  3330.1  107.55  4675.9  109.38  4826.4  107.72    4848   98.34
  4998.2   96.43  5091.6  108.41  5486.5  110.22  5593.8  101.46  5761.6  110.24
  5788.6  100.15  5829.6  111.43  6209.7  108.98  6617.8  108.89  6761.4  107.98
    6884  107.43  7115.3  106.89  7121.2  106.87  7431.2  105.88  8179.2  107.82
  8833.4   110.5  9386.2  108.59  9714.2  125.89 11132.3  125.16 11322.5  128.69
#Mann= 14 ,-1 , 0
   335.5     .11       0  4675.9     .15       0  4826.4     .09       0
  5091.6     .15       0  6209.7     .11       0  6617.8     .15       0
  6761.4     .11       0    6884     .15       0  7115.3     .11       0
  7121.2     .15       0  7431.2     .11       0  8179.2     .15       0
  8833.4     .11       0 11132.3    .125       0
#XS Ineff= 1 ,-1
     830  2729.7  119.57
Permanent Ineff=
       F
Bank Sta=4826.4,5091.6
XS Rating Curve= 0 ,0
Exp/Cntr=0.3,0.1

Type RM Length L Ch R = 1 ,231000  ,2000,2000,2000
BEGIN DESCRIPTION:
WFSJ Main 230.0
END DESCRIPTION:
XS GIS Cut Line= 3
      3843482.23     10089266.93      3840644.78     10085094.76
      3839560.36     10080766.96
#Sta/Elev= 30
   -45.6  145.64   723.7  123.55  1337.2  117.48  1855.1  120.79  2178.4  110.24
    2223  100.44  2259.1  110.41  2408.8  114.82  2480.7   109.2  3143.4  114.62
  3265.5  113.28  3291.4  113.29  3387.6  113.33  3623.6   113.8  3934.8  108.73
  4827.4  106.99  4835.2  105.54  4857.2   96.93  4998.2   96.01  5117.2   97.91
  5137.8  106.51  6416.7  107.02  6493.5  107.26  6575.1  107.61  7470.1  109.06
  7515.9  104.92  8224.8  109.26  8529.5  108.88  8828.5  125.78  9461.6  127.69
#Mann= 15 ,-1 , 0
   -45.6     .11       0  3143.4    .125       0  3265.5     .11       0
  3291.4    .125       0  3387.6     .11       0  3623.6     .17       0
  3934.8     .15       0  4827.4     .12       0  4835.2     .09       0
  5137.8     .15       0  6416.7     .11       0  6493.5     .15       0
  6575.1     .11       0  7470.1     .15       0  8224.8     .11       0
#XS Ineff= 1 ,-1
    1960  3049.4  114.81
Permanent Ineff=
       F
Bank Sta=4835.2,5137.8
XS Rating Curve= 0 ,0
Exp/Cntr=0.3,0.1

Type RM Length L Ch R = 1 ,229000  ,1361,1361,1361
BEGIN DESCRIPTION:
WFSJ Main 228.0
END DESCRIPTION:
XS GIS Cut Line= 3
      3844232.23     10088548.18      3842185.14      10084325.3
      3839732.55     10080720.52
#Sta/Elev= 30
   307.1  138.62   651.7  127.36  1415.2  114.59  1437.4  118.28  2209.1  116.07
  2598.4  104.49  3371.2  110.41  3859.1  106.16  3982.3    99.4  4031.8  105.29
  4589.1  104.26  4595.4   104.6  4707.3  104.04  4818.7  106.25  4844.2   96.07
  4998.2   94.32  5037.5  101.35  5088.3   94.82 5124.27  106.29  5151.3  110.48
  6058.2  106.09  6686.3  109.65  7153.5  104.99  7756.5  110.48  8045.5  109.21
  8269.9  121.53  8434.6  123.81  8859.5  122.01  9032.8  127.92    9360  127.83
#Mann= 10 ,-1 , 0
   307.1     .11       0  3371.2     .17       0  3859.1     .15       0
  4031.8     .17       0  4589.1     .15       0  4595.4     .17       0
  4707.3     .11       0  4818.7     .07       0 5124.27     .11       0
  7756.5     .11       0
Bank Sta=4818.7,5124.27
XS Rating Curve= 0 ,0
Exp/Cntr=0.3,0.1

Type RM Length L Ch R = 1 ,227639  ,2017,2017,2017
BEGIN DESCRIPTION:
WFSJ Main 227.0
END DESCRIPTION:
XS GIS Cut Line= 3
      3844857.23     10088345.05      3843107.22     10084470.05
      3840654.97     10080424.61
#Sta/Elev= 30
    1064  158.04  1904.2  113.99  2231.5  115.27  2275.7  115.34  3184.5  116.53
  3722.3  109.31  3832.1  109.26  3864.7  109.24  3982.2  109.18  4573.7     111
 4764.04106.1414  4769.6  105.32    4799   94.36  4998.2   93.82  5109.8  104.59
  5201.6  103.46  5373.1  102.88  5438.7  107.83  5692.8  104.17  5714.1  108.02
  6274.5  102.42  6305.4  107.33  6472.3  109.73    7463  108.79  7499.9  104.18
  7548.4  109.07  7965.1   111.2  9392.3  110.54  9603.7  122.69 10046.5  126.16
#Mann= 12 ,-1 , 0
    1064     .11       0  2231.5     .15       0  2275.7     .11       0
  3722.3     .15       0  3832.1     .11       0  3864.7     .15       0
  3982.2     .11       0 4764.04     .08       0  4769.6     .06       0
  5109.8     .11       0  5201.6     .15       0  7965.1     .11       0
Bank Sta=4769.6,5109.8
XS Rating Curve= 0 ,0
Exp/Cntr=0.3,0.1

Type RM Length L Ch R = 1 ,225622  ,1700,1700,1700
BEGIN DESCRIPTION:
WFSJ Main 225.0
END DESCRIPTION:
XS GIS Cut Line= 4
      3845529.12     10087938.83       3843654.1     10083235.67
      3843169.72     10082829.42      3840857.38     10079985.86
#Sta/Elev= 30
  -407.7  143.85   117.1  142.39   583.5  113.48  1872.1   116.2    2153   105.2
  2260.5  107.36  2602.5  105.22  2750.3  105.16    3013  105.95  3980.5  107.85
    4048  105.07  4387.3  105.59  4434.3  100.46    4585  105.02  4632.6   97.48
    4734  103.39  4805.5  102.23  4826.4   94.19  4918.7    98.3  4998.2   92.87
 5034.53  102.25  5081.4  107.85  6696.8   106.2  6995.5  109.89  7294.2  113.07
    7593  113.38  7790.8  111.96  7891.7  111.28  8301.5  124.11  8952.7  124.68
#Mann= 16 ,-1 , 0
  -407.7     .11       0    2153     .15       0  2260.5     .11       0
  2602.5     .15       0  2750.3     .11       0    3013     .15       0
  3980.5     .11       0    4048     .15       0    4734     .07       0
 5034.53     .15       0  6696.8     .17       0  6995.5     .11       0
  7294.2     .17       0    7593     .11       0  7790.8     .17       0
  7891.7     .11       0
#XS Ineff= 1 ,-1
     400  1872.1   116.2
Permanent Ineff=
       F
Bank Sta=4734,5034.53
XS Rating Curve= 0 ,0
Exp/Cntr=0.3,0.1

Type RM Length L Ch R = 1 ,223922  ,2476,2476,2476
BEGIN DESCRIPTION:
WFSJ Main 223.0
END DESCRIPTION:
XS GIS Cut Line= 5
      3845982.23     10087891.95      3844310.35     10083016.92
      3844372.85     10082360.67       3843966.6      10081563.8
       3840655.5       10077352.
#Sta/Elev= 30
 -1176.1   141.9  -873.5  139.64  -444.5  128.19    55.7  122.12    93.4  114.12
   211.1  113.81   379.9  112.28   727.1  112.68  1002.4  113.04  2001.8  108.66
  3701.7  106.43  4146.3  105.76  4532.4  105.39 4929.31  102.14  4950.7   92.36
  4998.2   91.36    5265   93.06 5301.55102.2279  5534.4  106.32  7156.2   110.1
  7277.4  113.14  7398.2   99.59  7483.2  110.71    7801  110.87  8874.9  109.87
  9228.3  107.17  9358.9  114.23  9997.9  122.17 10765.6  122.98 10888.8  124.54
#Mann= 20 ,-1 , 0
 -1176.1     .11       0  -873.5     .17       0  -444.5     .11       0
   211.1     .17       0   379.9     .17       0   727.1     .11       0
  1002.4     .11       0  2001.8     .15       0  3701.7     .11       0
  4146.3     .15       0  4532.4     .11       0 4929.31     .06       0
 5301.55     .11       0  5534.4     .15       0  7156.2     .11       0
    7801     .17       0  8874.9     .15       0  9358.9     .11       0
  9997.9     .11       0 10765.6     .11       0
#XS Ineff= 2 ,-1
  7263.5    9530  113.16      52  1228.2   114.3
Permanent Ineff=
       F       F
Bank Sta=4929.31,5301.55
XS Rating Curve= 0 ,0
Exp/Cntr=0.3,0.1

Type RM Length L Ch R = 1 ,221446  ,2446,2446,2446
BEGIN DESCRIPTION:
WFSJ Main 221.0
END DESCRIPTION:
XS GIS Cut Line= 3
      3851173.23      10086029.2      3844256.05     10080328.07
      3841685.61     10076640.22
#Sta/Elev= 30
 -2146.4  143.77 -1179.4  131.18  -683.6   122.9  -100.8  120.09   949.2  115.03
  2291.2  108.56  3266.7  106.28  3902.5  104.93 4752.45   102.8    4903  101.45
  4931.7   91.35  4998.2   89.81  5123.2   90.66  5151.9  102.77  5549.3    95.9
  5584.8  101.86  6190.2  102.51    6679  103.03  6714.2   91.54  6792.4   104.6
  7011.2  106.13  7712.2   109.2  8394.6   111.7  8472.3  104.87  8926.8  110.52
  9321.3  112.22 10055.3   119.7 10758.9   122.8 11232.3  123.01 11312.7  122.95
#Mann= 19 ,-1 , 0
 -2146.4     .17       0 -1179.4     .17       0  -683.6     .11       0
  -100.8     .15       0   949.2     .15       0  2291.2     .15       0
  3266.7     .17       0  3902.5     .11       0 4752.45     .09       0
  5151.9     .15       0  5584.8     .17       0  6190.2     .15       0
  7011.2     .17       0  7712.2     .11       0  8926.8     .17       0
  9321.3     .15       0 10055.3     .11       0 10758.9    .125       0
 11232.3    .125       0
Bank Sta=4752.45,5151.9
XS Rating Curve= 0 ,0
Exp/Cntr=0.3,0.1

Type RM Length L Ch R = 1 ,219000  ,2147,2147,2147
BEGIN DESCRIPTION:
WFSJ Main 219.0
END DESCRIPTION:
XS GIS Cut Line= 3
      3851789.73     10085772.11      3846049.65     10079579.71
      3843503.47     10075700.37
#Sta/Elev= 30
 -3443.6  142.15 -2698.3  127.83 -2090.2  114.57 -1586.3   111.9 -1110.2  111.54
  -817.3  108.54    1211  108.96  1292.3  109.23    1328  103.34  2092.7  108.33
  2539.5  110.73  2861.7  112.46    3953  108.37  4112.8  102.45  4165.6   97.43
  4264.2   97.66  4306.7  101.97  4505.2   98.04  4519.3  102.98    4599  102.44
  4887.3  102.01  4915.6   89.91  4998.2    88.7  5080.7   89.82 5115.74102.0369
  5240.8  103.06  6121.2  111.76  6762.9  121.66  7157.9  124.39  9640.3  121.85
#Mann= 17 ,-1 , 0
 -3443.6     .17       0 -2698.3     .17       0 -1586.3     .15       0
 -1110.2     .11       0  -817.3     .15       0    1211     .15       0
  2092.7     .17       0  2539.5     .11       0  2861.7     .17       0
  4112.8     .15       0    4599     .11       0  4887.3     .07       0
 5115.74     .11       0  5240.8     .17       0  6121.2     .11       0
  6762.9    .125       0  7157.9     .11       0
#XS Ineff= 1 ,-1
   -1750  2948.3  112.92
Permanent Ineff=
       F
Bank Sta=4887.3,5115.74
XS Rating Curve= 0 ,0
Exp/Cntr=0.3,0.1

Type RM Length L Ch R = 1 ,216853  ,1914,1914,1914
BEGIN DESCRIPTION:
WFSJ Main 217.0
END DESCRIPTION:
XS GIS Cut Line= 4
       3852119.6     10085615.87      3847711.62     10079799.91
       3847676.9     10079426.64      3844463.35     10075667.95
#Sta/Elev= 30
 -2501.7   138.7 -2261.1  139.98 -2225.8  137.42 -2204.9  125.77   -2154     128
 -2105.1  138.32 -1530.2  126.33    -446  105.79  -107.1   104.1   971.2  104.74
  1422.7  105.47  2459.7  103.98  3599.8  108.85    4845  100.23  4875.1   88.74
  4998.2    85.2 5060.66  100.93  5362.1   89.21    5642   86.73  5898.1   103.6
  6145.9   102.2  6300.5  115.68  6833.3  117.97  7282.5  117.51    7394  109.44
  8340.7  116.77  8839.5  118.24  9626.2  120.56 10055.6   123.7   10116  125.13
#Mann= 20 ,-1 , 0
 -2501.7     .11       0   -2154     .11       0 -1530.2     .17       0
    -446     .17       0  -107.1     .15       0   971.2     .15       0
  1422.7     .15       0  2459.7     .15       0  3599.8     .11       0
    4845     .07       0 5060.66     .15       0  5362.1     .11       0
  5898.1     .11       0  6300.5     .17       0  6833.3     .15       0
  7282.5     .17       0  8340.7     .11       0  8839.5    .125       0
  9626.2     .11       0 10055.6     .11       0
#XS Ineff= 1 ,-1
    -930  3577.4  110.03
Permanent Ineff=
       F
Bank Sta=4845,5060.66
XS Rating Curve= 0 ,0
Exp/Cntr=0.3,0.1

Type RM Length L Ch R = 1 ,214939  ,1939,1939,1939
BEGIN DESCRIPTION:
WFSJ Main 215.0
END DESCRIPTION:
XS GIS Cut Line= 3
      3852605.72     10085459.63      3849176.86     10079977.41
      3845105.73     10075251.31
#Sta/Elev= 30
 -1466.2  142.93 -1109.3  142.48  -465.7  141.77   -45.1  114.42   440.4     104
   926.8  105.29    1397   107.5  2676.9  102.81  4221.6   99.76  4879.6  105.73
  4910.2   95.38  4998.2   86.86  5131.2   88.03  5194.5   96.68  5251.9  103.37
  5495.8  100.99  6259.4  100.67    6337   100.9  6372.1   89.31  6414.9   99.34
  6748.4   97.31  6790.2  109.78  7059.8  116.43    7476  114.89  7953.1  108.19
  7979.9  112.62  8615.8  116.67 10244.2  123.15 10556.7  122.34 11237.8  123.72
#Mann= 18 ,-1 , 0
 -1466.2     .17       0 -1109.3     .17       0  -465.7     .11       0
   -45.1     .17       0   926.8     .11       0    1397     .17       0
  2676.9     .15       0  4221.6     .17       0  4910.2     .07       0
  5194.5     .17       0  5495.8     .15       0  6259.4     .11       0
  7059.8     .15       0    7476     .17       0  7979.9     .17       0
  8615.8     .15       0 10244.2    .125       0 10556.7    .125       0
Bank Sta=4910.2,5194.5
XS Rating Curve= 0 ,0
Exp/Cntr=0.3,0.1

Type RM Length L Ch R = 1 ,213000  ,2000,2000,2000
BEGIN DESCRIPTION:
WFSJ Main 213.0
END DESCRIPTION:
XS GIS Cut Line= 3
      3854322.64     10084948.48      3850210.22     10079093.76
      3847084.23     10074452.63
#Sta/Elev= 30
 -2154.7  146.89  -425.3  125.81      60  108.17   989.3   104.5  1426.9  105.78
  1813.4  104.46  2201.1   104.2  2661.7   103.9  2950.3  103.71  3029.6   95.51
  3044.4  103.96  3109.1  111.48  3487.1  104.89    3854  103.04  4917.7  102.33
 4936.3795.71989  4945.8    88.6  4998.2   86.17  5242.1   95.03  5320.1    88.6
  5392.1  100.63  5455.1   98.27    5494   92.88    6103  103.17  7076.5  110.23
    8237   112.5  9510.4  116.79  9997.2  117.75 10510.1  120.45 10595.7   120.9
#Mann= 19 ,-1 , 0
 -2154.7     .11       0  -425.3     .17       0      60     .11       0
   989.3     .17       0  1426.9     .17       0  1813.4     .15       0
  2201.1     .15       0  2661.7     .17       0  3487.1     .17       0
    3854     .15       0 4936.37     .07       0  5242.1     .15       0
  5455.1     .17       0    6103     .15       0  7076.5     .11       0
    8237     .17       0  9510.4    .125       0  9997.2    .125       0
 10510.1     .11       0
#XS Ineff= 1 ,-1
    -200  3109.1  111.48
Permanent Ineff=
       F
Bank Sta=4936.37,5242.1
XS Rating Curve= 0 ,0
Exp/Cntr=0.3,0.1

Type RM Length L Ch R = 1 ,211000  ,1747,1747,1747
BEGIN DESCRIPTION:
WFSJ Main 211.0
END DESCRIPTION:
XS GIS Cut Line= 3
      3855115.47     10084685.26      3851087.52     10077597.56
      3847257.87     10074181.39
#Sta/Elev= 30
 -3152.3  138.83 -2544.7  141.61 -2357.6  141.87 -1866.7  140.96 -1470.5  138.11
 -1246.4  118.09 -1082.7   107.5  -684.3  105.22  -259.4  103.56   -18.9  107.86
   222.6   98.99   392.1  107.66   602.6   97.99  1310.4   99.85  1502.4  100.36
  1735.3  100.97  4512.1   97.52  4887.3  100.48 4916.38   93.03  4998.2   85.35
 5136.0693.39973  5712.4  109.88  7706.5  111.86  8010.9  112.31  8538.9  110.36
    8986  114.35  9191.8  115.64  9779.5  116.93 10057.6  121.28 10131.9     122
#Mann= 20 ,-1 , 0
 -3152.3     .11       0 -2544.7     .11       0 -2357.6     .17       0
 -1866.7     .11       0 -1246.4     .11       0  -684.3     .15       0
  -259.4     .15       0  1310.4     .17       0  1502.4     .11       0
  1735.3     .15       0  4512.1     .12       0 4916.38     .07       0
 5136.06     .12       0  7706.5     .17       0  8010.9     .11       0
  8538.9    .125       0    8986     .15       0  9191.8    .125       0
  9779.5     .11       0 10057.6     .11       0
#XS Ineff= 1 ,-1
   -1170   392.1  107.66
Permanent Ineff=
       F
Bank Sta=4916.38,5136.06
XS Rating Curve= 0 ,0
Exp/Cntr=0.3,0.1

Type RM Length L Ch R = 1 ,209253  ,2253,2253,2253
BEGIN DESCRIPTION:
WFSJ Main 209.0
END DESCRIPTION:
XS GIS Cut Line= 3
      3855365.48     10084497.78      3852282.15      10076143.6
      3847323.85     10074101.95
#Sta/Elev= 30
 -3538.5  131.62 -3217.5  136.54 -2461.2  140.82   -2217  133.04 -1697.6  127.86
 -1468.8  108.49 -1368.8  101.48  -772.2  106.67  -318.8  104.03   -23.5  107.85
   272.3  103.73   677.9  105.46  1398.2  101.84  1673.2  100.73  2126.6   92.84
  2414.9  102.34  3800.9  100.67  4150.1   87.77    4218   97.45  4449.8   96.88
  4843.1   92.69  4998.1    84.5    5156    92.5  5192.3  100.88  6010.6  104.96
  6577.1  110.94  9395.8  114.68 10360.1   118.7 10674.9  121.47 10728.7  121.69
#Mann= 20 ,-1 , 0
 -3538.5     .11       0 -3217.5     .17       0   -2217     .11       0
 -1697.6     .17       0 -1468.8     .15       0  -772.2     .17       0
  -318.8     .15       0   -23.5     .17       0   272.3     .15       0
   677.9     .15       0  1398.2     .11       0  1673.2     .15       0
  4449.8     .17       0  4843.1     .09       0    5156     .17       0
  6010.6     .11       0  6577.1     .11       0  9395.8    .125       0
 10360.1    .125       0 10674.9     .11       0
#XS Ineff= 1 ,-1
   -1550   583.2  108.05
Permanent Ineff=
       F
Bank Sta=4843.1,5156
XS Rating Curve= 0 ,0
Exp/Cntr=0.3,0.1

Type RM Length L Ch R = 1 ,207000  ,1726,1726,1726
BEGIN DESCRIPTION:
WFSJ Main 207.0
END DESCRIPTION:
XS GIS Cut Line= 4
      3855636.32      10084372.8       3854336.8     10077258.52
      3853157.15      10075643.6      3847293.06     10074061.65
#Sta/Elev= 30
   -2232  124.76 -2179.4  121.37 -2125.5  129.68  -821.9   136.1  -705.2  133.25
  -465.6  109.87     9.5  104.99  1218.7  105.08  1553.8  106.59  2362.9   103.4
  3237.9  101.78  3916.5  102.17  4824.6   99.27 4860.97   92.26  4998.1   83.15
  5161.6    84.4    5191   92.56  5326.9   95.73    5513   97.62  5584.1   90.67
    5716   98.69  6071.4  100.32  6284.8   93.13  7091.7  101.01  7808.8  103.41
  8335.4  105.14 11855.8  114.66 12199.3  115.28 12970.6  121.33 13073.6  121.96
#Mann= 20 ,-1 , 0
   -2232    .125       0 -2125.5     .17       0  -465.6     .15       0
     9.5     .15       0  1218.7     .17       0  1553.8     .15       0
  2362.9     .17       0  3237.9     .15       0  3916.5     .15       0
 4860.97     .09       0    5191     .15       0  5326.9     .11       0
    5716     .11       0  6284.8     .15       0  7091.7     .11       0
  7808.8     .15       0  8335.4     .11       0 11855.8     .15       0
 12199.3    .125       0 12970.6     .11       0
#XS Ineff= 1 ,-1
    -550  2008.8   108.1
Permanent Ineff=
       F
Bank Sta=4860.97,5191
XS Rating Curve= 0 ,0
Exp/Cntr=0.3,0.1

Type RM Length L Ch R = 1 ,205274  ,1136,1136,1136
BEGIN DESCRIPTION:
WFSJ Main 205.0
END DESCRIPTION:
XS GIS Cut Line= 3
      3858851.43      10078655.9      3854844.44     10075736.28
      3847362.32     10074017.65
#Sta/Elev= 30
   867.9  149.15  1818.7  125.08  2333.3  108.35  2387.5  100.12  2553.6   92.93
  2633.2  104.87  2877.2   99.49  3389.3  103.97  3659.3  104.56  4632.5  104.34
  4818.7  103.17  4845.7   90.95  4868.8   83.08  4998.1   82.27  5211.9   90.06
  5326.6   84.49  5483.9   95.99  5684.7    97.8  6150.6   92.73    6271  106.35
  6524.7  102.57  6903.8  101.89  7419.6  101.87  7594.5  101.87  8414.1  100.75
 12252.1  117.63 12422.7  117.54 12660.9  118.06 12739.8  118.51 13502.7  120.74
#Mann= 19 ,-1 , 0
   867.9     .17       0  2387.5     .11       0  2553.6     .15       0
  2633.2     .17       0  3389.3     .11       0  3659.3     .17       0
  4632.5     .11       0  4845.7     .06       0  5211.9     .11       0
    6271     .15       0  6524.7     .17       0  6903.8     .15       0
  7419.6     .17       0  7594.5     .15       0  8414.1     .11       0
 12252.1    .125       0 12422.7     .15       0 12660.9    .125       0
 12739.8     .11       0
Bank Sta=4845.7,5211.9
XS Rating Curve= 0 ,0
Exp/Cntr=0.3,0.1

Type RM Length L Ch R = 1 ,204138  ,648,648,648
BEGIN DESCRIPTION:
WFSJ Main 204.0
END DESCRIPTION:
XS GIS Cut Line= 4
      3859426.04     10077101.67      3855389.56     10075267.89
      3853067.51     10074378.14      3847197.27     10073987.51
#Sta/Elev= 30
   335.6  126.24   597.2  108.54    1190  104.04  2071.6  103.08  2629.2  101.89
    2728   84.21  2787.5   87.89  2835.9   103.1  4278.6  101.66    4579  100.59
  4835.3  101.79  4867.3   91.64  4998.1   81.87  5108.9   92.35  5574.1   89.55
  5747.3  103.65    6509  112.13  6533.7  102.61  6679.8  103.44  7040.6   106.9
  7406.7  104.01  7677.9  103.53  7897.9  102.46  8292.3  100.72 10329.6  118.47
 11459.7  119.93 11860.6   118.6 12080.8  119.32 13025.7   122.4   13139  122.77
#Mann= 20 ,-1 , 0
   335.6     .17       0    1190     .17       0  2071.6     .11       0
  2787.5     .17       0  4278.6     .17       0    4579     .15       0
  4867.3     .09       0  5108.9    .125       0  5747.3     .11       0
  6679.8    .125       0  7040.6     .11       0  7406.7    .125       0
  7677.9     .11       0  7897.9     .15       0  8292.3     .11       0
 10329.6     .11       0 11459.7    .125       0 11860.6    .125       0
 12080.8     .11       0 13025.7     .17       0
#Block Obstruct= 1 ,-1
    6509    9950  112.13
Bank Sta=4867.3,5108.9
XS Rating Curve= 0 ,0
Exp/Cntr=0.3,0.1

Type RM Length L Ch R = 1 ,203490  ,1564,1564,1564
BEGIN DESCRIPTION:
WFSJ Main 203.0
END DESCRIPTION:
XS GIS Cut Line= 6
      3859498.83     10076891.05       3856995.4     10075759.13
      3855849.56     10075168.85      3855863.45     10075043.85
      3853241.12     10073824.75      3847284.08     10073640.29
#Sta/Elev= 30
  -173.9   136.3  -155.6   135.6   111.2  110.42   430.4  105.12  1668.8  104.44
  2208.7  101.85  2274.5   82.17  2526.9   99.29  3211.7   96.91  3482.9  100.28
  4160.4    98.6  4691.2   95.22 4704.83   92.46  4998.1   81.43 5027.9592.55892
  5780.6   87.52  6113.9  101.68  6517.7     106  6574.9    89.9  6854.7   99.96
  7113.5   86.36  7181.6   97.65  8745.4  107.51  8955.9  108.78  9251.6  110.57
  9718.6  118.46  9941.6  118.93 12307.4  122.68 12701.7  123.31   12840  123.53
#Mann= 20 ,-1 , 0
  -173.9     .11       0  -155.6    .125       0   111.2    .125       0
   430.4    .125       0  1668.8    .125       0  3211.7     .11       0
  3482.9    .125       0  4160.4    .125       0  4691.2     .15       0
 4704.83     .09       0 5027.95    .125       0  6113.9    .125       0
  7181.6     .15       0  8745.4    .125       0  8955.9     .17       0
  9251.6    .125       0  9718.6    .125       0  9941.6     .11       0
 12307.4     .11       0 12701.7     .17       0
#Block Obstruct= 2 ,-1
      38  1581.7  110.96  6517.7    8560     106
Bank Sta=4704.83,5027.95
XS Rating Curve= 0 ,0
Exp/Cntr=0.3,0.1

Type RM Length L Ch R = 1 ,201926  ,1092,1092,1092
BEGIN DESCRIPTION:
WFSJ Main 202.0
END DESCRIPTION:
XS GIS Cut Line= 4
      3861250.82     10076007.56      3856276.84     10074106.51
      3855977.36     10073637.76      3847111.54     10072088.52
#Sta/Elev= 30
  -579.6  146.71   239.3  102.82   592.7  102.24   956.9  101.65  1231.5   101.2
  1577.9  101.98  3984.1  108.36  4091.2   87.54  4929.7   90.63  4998.1   75.76
 5465.91   90.87  5572.6  100.35  5834.1   83.71  6316.6   87.48  6567.4   95.28
  7064.8   89.04  7345.6   82.96  7412.6  100.55    7443   81.84  7548.2   88.48
  7762.3   89.53  7973.8   95.14  8217.8  110.37 10082.4  102.53 11787.9  113.68
 11820.6  125.72 11975.9  116.41 12595.5  117.95 14060.4  120.34 14301.7  118.38
#Mann= 18 ,-1 , 0
  -579.6     .17       0   239.3     .15       0   592.7     .17       0
   956.9     .17       0  1231.5     .11       0  1577.9     .11       0
  4929.7     .07       0 5465.91     .11       0  5572.6     .15       0
  6316.6     .11       0  6567.4     .15       0  7064.8     .11       0
  7548.2     .15       0  7762.3     .15       0  7973.8     .11       0
 11975.9     .17       0 12595.5     .11       0 14060.4     .15       0
#Block Obstruct= 3 ,-1
  8217.8   11245  110.37     -65  1835.6  112.94    1836  3984.1  108.36
Bank Sta=4929.7,5465.91
XS Rating Curve= 0 ,0
Exp/Cntr=0.3,0.1

Type RM Length L Ch R = 1 ,200834  ,834,834,834
BEGIN DESCRIPTION:
WFSJ Main 201.0
END DESCRIPTION:
XS GIS Cut Line= 4
       3862891.4     10074575.25      3856537.25     10073169.01
      3854308.11     10072459.15      3847344.56     10071997.13
#Sta/Elev= 30
 -1219.5   150.3  -580.9  103.25   902.3   99.53    1410   99.49  1601.6   99.48
  1735.2   99.47  2108.4   99.44  2128.4   99.44  2288.2   99.43  3842.5   99.32
  4898.6   90.45  4998.1   74.78  5074.2    76.1 5102.29   91.22  5676.1   99.23
  5987.5   91.24  6337.9   89.96  7371.7  100.32  8740.5   99.74  8780.6     114
  9281.7  115.73  9522.3  103.35 10263.9  113.12 10424.2   98.06 10835.1  110.99
 10915.3   98.75 12915.8   108.2 13184.3  118.28 14466.2   118.5 14606.7  118.42
#Mann= 18 ,-1 , 0
 -1219.5     .11       0   902.3     .17       0    1410     .15       0
  1601.6     .17       0  1735.2     .15       0  2108.4     .17       0
  2128.4     .15       0  2288.2     .17       0  3842.5     .15       0
  4898.6     .07       0 5102.29     .12       0  5676.1     .15       0
  5987.5     .11       0  6337.9     .15       0  7371.7     .11       0
 12915.8     .17       0 13184.3     .11       0 14466.2     .17       0
#Block Obstruct= 2 ,-1
  7340.4    9085  109.47  9281.7   13100  115.73
Bank Sta=4898.6,5102.29
XS Rating Curve= 0 ,0
Exp/Cntr=0.3,0.1

Type RM Length L Ch R = 1 ,200000  ,1000,1000,1000
BEGIN DESCRIPTION:
WFSJ Main 200.0
END DESCRIPTION:
XS GIS Cut Line= 4
      3863099.79     10073963.29      3856738.23     10072412.29
      3855026.84     10072049.22      3847474.75     10071814.84
#Sta/Elev= 30
 -1547.9  149.31  -578.4   99.71   -25.9  103.03   578.7    98.4   780.5   99.09
  1224.5   98.45  1752.2   98.88  2099.3  100.14  3149.5   98.91  3383.5   98.87
  4091.5   94.36  4619.9   98.82 4774.02  98.549 4801.97   91.37  4998.1   74.26
  5315.6   91.35  5863.3   89.24  6042.8   89.05  6848.8   90.31    7159   89.73
  7288.7  109.43    7585   101.9  8142.2  109.44  8299.2   95.12  9169.6  113.78
   11961   98.07 12611.3  118.39 12721.3  104.34   14288   119.4 14305.2  117.17
#Mann= 20 ,-1 , 0
 -1547.9     .11       0   -25.9     .17       0   578.7     .15       0
   780.5     .17       0  1224.5     .15       0  1752.2     .15       0
  2099.3     .17       0  3149.5     .17       0  3383.5     .15       0
  4091.5     .17       0  4619.9     .15       0 4774.02     .11       0
 4801.97     .06       0  5315.6     .11       0  5863.3     .11       0
  6042.8     .15       0  6848.8     .11       0    7159     .15       0
    7585     .11       0   14288     .17       0
#Block Obstruct= 2 ,-1
  7338.8    9066  109.18  9169.6   13127  113.78
Bank Sta=4801.97,5315.6
XS Rating Curve= 0 ,0
Exp/Cntr=0.3,0.1

Type RM Length L Ch R = 1 ,199000  ,1000,1000,1000
BEGIN DESCRIPTION:
WFSJ Main 199.0
END DESCRIPTION:
XS GIS Cut Line= 3
      3863568.51     10073142.97      3856608.15     10071429.79
      3849506.01      10070603.9
#Sta/Elev= 30
 -2168.1  140.79  -709.6  129.69  -381.3  125.78   174.8   98.07  2711.6   98.48
  3321.7   89.08  3593.8   96.52  3635.3   88.47    3713   95.07  4528.3    97.3
  4725.1   99.78 4790.34   91.56  4835.5   75.47  4998.1   74.42  5161.4   85.86
  5312.4   78.69 5351.43   91.73  5372.8   99.27  5718.7   100.2  6802.8   99.37
  6953.1   94.54  7033.9     105  7758.8  101.85  8030.6  112.03  8070.8   95.01
    9138   95.47  9362.7  113.89  9812.5  112.52  9962.7  104.19   12150  121.84
#Mann= 11 ,-1 , 0
 -2168.1     .11       0  -709.6     .17       0   174.8     .15       0
  4528.3     .17       0  4725.1     .11       0 4790.34     .07       0
 5351.43     .11       0  5372.8     .15       0  5718.7     .11       0
  6802.8     .15       0  6953.1     .11       0
#Block Obstruct= 1 ,-1
  8030.6   10640  112.03
Bank Sta=4790.34,5351.43
XS Rating Curve= 0 ,0
Exp/Cntr=0.3,0.1

Type RM Length L Ch R = 1 ,198000  ,1761,1761,1761
BEGIN DESCRIPTION:
WFSJ Main 198.0
END DESCRIPTION:
XS GIS Cut Line= 5
      3863724.79     10072791.41      3856913.52     10070661.55
      3855847.15     10069861.72      3854675.27     10068598.69
      3852762.04     10067817.78
#Sta/Elev= 30
 -2136.5  131.72 -1825.4  118.73   -12.8   125.2   410.7  106.51   819.4  104.88
   921.5  104.46  1149.3  103.53  3846.9   86.63  4041.7      99  4117.1    85.4
  4673.5   91.28  4998.1   74.13    5155   75.17  5182.1   91.02    5205   93.99
  5346.6   92.77  5382.1   82.34  5669.6  101.13  5816.4   86.67  6090.4   86.35
  6161.7  106.06  6207.1  109.43  7168.5  115.59  7301.2   116.7  7446.7  117.14
  7585.8  117.34  7731.6  118.32    8099  119.04  9668.8  118.27 10122.4     124
#Mann= 18 ,-1 , 0
 -2136.5     .11       0   410.7     .17       0   819.4     .15       0
   921.5     .17       0  1149.3     .15       0  4673.5     .07       0
  5182.1     .11       0    5205     .15       0  5816.4     .11       0
  6161.7     .17       0  6207.1     .11       0  7168.5     .17       0
  7301.2     .11       0  7446.7    .125       0  7585.8     .11       0
  7731.6    .125       0    8099     .11       0  9668.8     .17       0
Bank Sta=4673.5,5182.1
XS Rating Curve= 0 ,0
Exp/Cntr=0.3,0.1

Type RM Length L Ch R = 1 ,196239  ,1239,1239,1239
BEGIN DESCRIPTION:
WFSJ Main 196.0
END DESCRIPTION:
XS GIS Cut Line= 3
      3864128.43     10072309.64      3858672.67     10069991.92
      3852904.43     10067570.04
#Sta/Elev= 30
 -1248.1     147   -1195  146.77  -888.9  147.64   110.6  115.05   474.6  108.91
  1735.8  103.73  2579.1  104.17  3904.5   94.88  4101.7   94.39  4852.7   94.17
  4898.8   95.59  4933.489.29115  4998.1   73.66  5216.5   77.75 5242.9289.42747
    5264   91.74  5287.8   80.28  5316.9   86.88  5499.5   88.09  5547.1   98.02
  5629.2   96.32  6888.5   98.85  7513.5  104.59  8076.3  116.52  8530.9  117.72
  8570.9   118.1  8771.6  119.81  8949.3  119.72  9889.7  115.36 10935.6  118.08
#Mann= 17 ,-1 , 0
 -1248.1     .17       0   -1195     .11       0  1735.8     .17       0
  2579.1     .15       0  3904.5     .17       0  4101.7     .15       0
  4852.7     .11       0  4933.4     .07       0 5242.92     .15       0
  5629.2     .15       0  6888.5     .17       0  7513.5     .11       0
  8530.9    .125       0  8570.9     .11       0  8771.6    .125       0
  8949.3     .11       0  9889.7     .17       0
Bank Sta=4933.4,5242.92
XS Rating Curve= 0 ,0
Exp/Cntr=0.3,0.1

Type RM Length L Ch R = 1 ,195000  ,1508,1508,1508
BEGIN DESCRIPTION:
WFSJ Main 195.0
END DESCRIPTION:
XS GIS Cut Line= 3
      3864948.68     10071307.02      3858877.01      10068844.6
      3852995.59     10067270.57
#Sta/Elev= 30
   -1552  136.13 -1250.8  137.78  -422.3  130.37   416.3   118.5   786.7  113.26
  1464.6  103.57  2176.4  104.93  2344.5   88.84  2398.4  101.51    2474   88.58
  2516.6   97.71  2551.5   88.67  2617.7  104.76  2830.1   110.4  2945.1  100.49
  3314.8  104.73  3598.3  101.84  4434.9   96.69  4713.6   81.16  4863.6   90.08
  4880.4    86.4  4998.1   72.67    5144   76.27    5184   86.76  5229.2   97.33
  6442.8   95.17  6879.2   96.29  7436.3   97.71  7653.4   98.27 11088.4  116.18
#Mann= 19 ,-1 , 0
   -1552     .11       0 -1250.8     .17       0  -422.3     .17       0
   416.3     .15       0   786.7     .11       0  1464.6     .11       0
  2617.7     .15       0  2945.1     .11       0  3314.8     .17       0
  3598.3     .15       0  4434.9     .17       0  4713.6     .15       0
  4863.6     .11       0  4880.4     .07       0    5184     .17       0
  6442.8     .15       0  6879.2     .11       0  7436.3     .17       0
  7653.4     .11       0
#Block Obstruct= 1 ,-1
     940  3165.1  108.68
Bank Sta=4880.4,5184
XS Rating Curve= 0 ,0
Exp/Cntr=0.3,0.1

Type RM Length L Ch R = 1 ,193492  ,1492,1492,1492
BEGIN DESCRIPTION:
WFSJ Main 193.0
END DESCRIPTION:
XS GIS Cut Line= 3
      3865722.57     10070226.73      3859993.42     10067791.84
      3853274.66     10066086.11
#Sta/Elev= 30
 -1505.4   144.8  -639.9  119.32  -287.5  117.57  1575.1  102.51  2306.9  105.81
  2354.2  121.61  2389.6   112.8  2422.2   87.88  2712.4   87.42  2900.3  108.74
  2965.2   99.31  3663.5  107.66  3693.5   99.07  4911.2   88.37  4921.5   83.44
  4998.1   70.73  5228.3   83.75  5406.4   83.79  5438.2    97.1  5716.2   96.39
    6452   96.01  6754.4   95.82    6956   98.46  8770.3   96.86  9759.6   98.97
 10067.8   98.71 10366.8    98.3 10478.3  108.83 10612.2  113.37 11651.6  114.72
#Mann= 18 ,-1 , 0
 -1505.4     .11       0  -639.9     .15       0  -287.5     .11       0
  1575.1     .11       0  4911.2     .11       0  4921.5     .07       0
  5228.3     .11       0  5406.4     .17       0  5716.2     .15       0
    6452     .11       0  6754.4     .17       0    6956     .15       0
  8770.3     .11       0  9759.6     .17       0 10067.8     .15       0
 10366.8     .17       0 10478.3     .11       0 10612.2     .17       0
#Block Obstruct= 2 ,-1
    2376  3663.5  107.66    -900  2354.2  121.61
Bank Sta=4921.5,5228.3
XS Rating Curve= 0 ,0
Exp/Cntr=0.3,0.1

Type RM Length L Ch R = 1 ,192000  ,2000,2000,2000
BEGIN DESCRIPTION:
WFSJ Main 192.0
END DESCRIPTION:
XS GIS Cut Line= 3
      3867024.66     10068338.71      3860434.33     10066448.65
      3853601.49     10065226.96
#Sta/Elev= 30
   -1856  137.15  -687.3  109.25     3.4  109.67   262.6  104.59  1238.2  101.84
  1647.3  101.38  2301.9  106.53  2755.9   94.71  2998.9   95.32    3680   95.62
  4714.7   93.36  4753.6   83.42  4809.1   73.11  4998.1   69.93    5067   71.83
 5094.0584.61525  5130.9   96.26  5219.9   87.43  6094.3   95.31  6506.7    94.7
  7203.4   99.64  7601.5      99  9424.2   95.56  9780.3   96.06 10217.9   96.84
 10467.9  114.64 10686.8  116.86 11283.9  114.67 11929.6  114.91 11941.2  114.91
#Mann= 19 ,-1 , 0
   -1856     .11       0     3.4     .15       0   262.6     .11       0
  1238.2     .15       0  1647.3     .11       0  2755.9     .11       0
  2998.9     .15       0    3680     .11       0  4753.6     .07       0
 5094.05     .17       0  6094.3     .15       0  6506.7     .11       0
  7203.4     .17       0  7601.5     .15       0  9424.2     .11       0
  9780.3     .15       0 10686.8     .11       0 11283.9     .11       0
 11929.6     .15       0
Bank Sta=4753.6,5094.05
XS Rating Curve= 0 ,0
Exp/Cntr=0.3,0.1

Type RM Length L Ch R = 1 ,190000  ,2000,2000,2000
BEGIN DESCRIPTION:
WFSJ Main 190.0
END DESCRIPTION:
XS GIS Cut Line= 3
      3867805.92       10066646.      3859938.21     10064731.89
       3854055.9     10063312.67
#Sta/Elev= 30
 -3097.2  133.01 -2292.5  123.89 -1882.7  102.72  -737.1   99.44  -440.6   97.06
    23.5   96.16  1118.3   95.87  1625.1   94.29  2172.3   94.06  3158.6   95.22
  3536.2   94.48  3757.9   86.39  3847.7   95.39  4441.5   93.75  4763.7   94.57
 4792.18   85.27  4998.1   69.66  5109.2   70.16  5156.8   85.71  5185.5   94.54
  5407.6   97.01  6605.1   98.66    7257   99.08  7531.3   95.55  9050.1   97.52
  9444.3   98.02    9627  115.85 10258.5  113.66 10609.2  113.43 11051.1  113.78
#Mann= 19 ,-1 , 0
 -3097.2     .11       0 -1882.7     .17       0  -737.1     .15       0
  -440.6     .11       0    23.5     .15       0  1118.3     .15       0
  1625.1     .11       0  2172.3     .11       0  3158.6     .15       0
  3536.2     .15       0  4441.5     .11       0 4792.18     .07       0
  5156.8     .17       0  6605.1     .15       0    7257     .11       0
  7531.3     .15       0  9050.1     .15       0 10258.5     .17       0
 10609.2     .11       0
Bank Sta=4792.18,5156.8
XS Rating Curve= 0 ,0
Exp/Cntr=0.3,0.1

Type RM Length L Ch R = 1 ,188000  ,2000,2000,2000
BEGIN DESCRIPTION:
WFSJ Main 188.0
END DESCRIPTION:
XS GIS Cut Line= 3
      3868144.44     10065682.46       3860889.5     10063124.74
      3855111.68     10061047.43
#Sta/Elev= 30
 -2692.6  131.01 -2347.1  121.12 -1969.2  126.82 -1625.5  106.32   -1392   93.73
  2210.8   96.11  2832.3   94.14  4119.9   92.93  4158.4   92.66  4212.9   92.28
  4249.2   81.83  4578.9   81.18  4998.1   68.59  5097.4   70.06 5137.6381.74817
  5175.2   92.74  6468.2   94.47  6723.3  100.67  6918.6   95.18    6944  100.14
  7276.6    97.8  7307.7  105.37  7388.8   97.52  7864.4   99.98  7920.5   94.21
  8051.6  104.48  8124.9   96.31  8723.3  112.09 11109.1   115.2 11139.9  115.31
#Mann= 10 ,-1 , 0
 -2692.6     .11       0 -1969.2     .17       0 -1625.5     .11       0
  2210.8     .15       0  2832.3     .11       0  4119.9     .17       0
  4158.4     .11       0  4578.9     .06       0 5137.63     .11       0
 11109.1     .17       0
Bank Sta=4578.9,5137.63
XS Rating Curve= 0 ,0
Exp/Cntr=0.3,0.1

Type RM Length L Ch R = 1 ,186000  ,2000,2000,2000
BEGIN DESCRIPTION:
WFSJ Main 186.0
END DESCRIPTION:
XS GIS Cut Line= 3
      3868717.39     10064367.36      3861339.03     10061731.95
      3855475.21     10060669.45
#Sta/Elev= 30
 -2834.9  124.02 -1400.3  127.39  -669.2   93.51  1330.9    94.6  1473.1   92.77
  2156.7   94.98  2260.9   92.47  3160.3   94.02  3985.9   94.56  4293.8   93.47
  4485.7   93.16  4696.7   84.89 4709.97   78.36  4998.1   67.18  5072.3   68.13
  5088.3   78.89  5141.8   89.45  5447.3   91.23  5853.6   87.64  6773.1   88.94
    6922  110.32  7167.6  123.24  7318.3   111.6  8035.8  112.29  8135.4  112.01
 10167.4  114.09 10325.6  114.59 10524.7  113.92 10798.1  111.97 10959.3  112.07
#Mann= 20 ,-1 , 0
 -2834.9     .11       0  1330.9     .15       0  1473.1     .15       0
  2156.7     .15       0  2260.9     .11       0  3160.3     .15       0
  3985.9     .17       0  4293.8     .15       0  4485.7     .15       0
  4696.7     .11       0 4709.97     .07       0  5088.3     .11       0
  5447.3    .125       0  5853.6     .11       0  8035.8    .125       0
  8135.4     .11       0 10167.4     .17       0 10325.6     .11       0
 10524.7     .15       0 10798.1     .17       0
Bank Sta=4709.97,5088.3
XS Rating Curve= 0 ,0
Exp/Cntr=0.3,0.1

Type RM Length L Ch R = 1 ,184000  ,1109,1109,1109
BEGIN DESCRIPTION:
WFSJ Main 184.0
END DESCRIPTION:
XS GIS Cut Line= 3
       3868899.7      10063885.6      3860787.93     10059997.15
      3855917.93     10059380.38
#Sta/Elev= 30
 -3995.6  117.08  -345.8  100.13   -23.5   99.62      84   99.21   191.4   98.97
   254.2   98.83   298.8   98.73   728.5   95.43  1519.4   89.78  3192.5   76.06
  3226.2   92.56    3481  103.92  3843.9   91.63  4058.7   90.46  4313.3   77.62
  4375.7   89.17  4398.4   78.68  4501.1   72.51  4778.778.74182  4998.1   66.09
  5080.7   67.16 5097.55   79.22    5121   97.36  6038.3   87.43  6764.3    88.6
  6844.7   98.71  6874.9   88.68  6999.6   90.59  7036.2   105.3  9908.9  111.85
#Mann= 14 ,-1 , 0
 -3995.6     .11       0  -345.8     .15       0   -23.5     .17       0
      84     .15       0   191.4     .17       0   254.2     .15       0
   298.8     .17       0   728.5     .15       0  1519.4     .11       0
  3843.9     .17       0  4058.7     .11       0  4375.7     .08       0
  4778.7     .06       0 5097.55     .11       0
#XS Ineff= 1 ,-1
    5121    7150   97.36
Permanent Ineff=
       F
#Block Obstruct= 1 ,-1
   -1700    3481  103.92
Bank Sta=4778.7,5097.55
XS Rating Curve= 0 ,0
Exp/Cntr=0.3,0.1

Type RM Length L Ch R = 1 ,182891  ,1695,1695,1695
BEGIN DESCRIPTION:
WFSJ Main 183.0
END DESCRIPTION:
XS GIS Cut Line= 4
      3869094.97     10063677.25      3861764.25     10059679.86
      3860996.02     10058859.55      3856165.28     10058182.46
#Sta/Elev= 30
 -3768.4  114.57 -2431.2  124.04  -626.2  100.68  -327.4    98.1   302.9   96.73
   648.9   95.98  1060.8   95.08  1317.8   94.52  2218.7    91.3  2706.5   89.71
  2777.7  100.41  3324.4   94.44  3392.7   83.03  4172.2      90  4201.4   81.37
  4466.5   81.72  4510.2   93.62  4627.5   94.33  4733.5   76.43  4938.6   78.74
  4998.1   65.65  5143.8   66.17 5191.98   78.38  5214.6   91.03  5264.4   91.49
  7089.7   96.31  7201.7   95.68  7254.4   95.41  7974.9  101.83 10583.2  109.98
#Mann= 16 ,-1 , 0
 -3768.4     .11       0  -626.2     .17       0  -327.4     .15       0
   302.9     .17       0   648.9     .15       0  1060.8     .17       0
  1317.8     .15       0  2218.7     .11       0  4627.5     .08       0
  4938.6     .06       0 5191.98     .08       0  5264.4     .11       0
  7089.7     .17       0  7201.7     .11       0  7254.4     .17       0
  7974.9     .11       0
#XS Ineff= 1 ,-1
    6804    7575   97.49
Permanent Ineff=
       F
#Block Obstruct= 2 ,-1
    -815  2777.7  100.41  2777.8  4548.1   95.41
Bank Sta=4938.6,5191.98
XS Rating Curve= 0 ,0
Exp/Cntr=0.3,0.1

Type RM Length L Ch R = 1 ,181196  ,2196,2196,2196
BEGIN DESCRIPTION:
WFSJ Main 182.0
END DESCRIPTION:
XS GIS Cut Line= 4
      3869719.95     10062791.82      3863730.39     10058794.44
      3863144.46     10059067.88      3858418.79     10054009.12
#Sta/Elev= 30
 -3096.9  116.94 -2908.5  115.98 -2401.4   113.4 -1938.3  111.04  -549.1   99.22
  -100.5  107.69   515.8  103.42  1217.3   91.51  1629.9   98.87  1745.4   97.96
  2208.1   94.33    2682   87.04  2999.5   91.13  3818.7   91.25  4486.9   78.07
  4526.2   90.19  4750.7   91.31  4809.7   80.37  4998.1   64.65  5262.6   80.81
  7065.4   91.09  7257.7   91.33  7292.9   80.54  7549.2   91.26  8328.8   95.53
  8468.5   96.29  8816.1   98.19 11026.7   110.5 11207.4  110.38 11673.3  108.97
#Mann= 20 ,-1 , 0
 -3096.9     .17       0 -2908.5     .11       0 -2401.4     .17       0
 -1938.3     .15       0  -100.5     .17       0   515.8     .15       0
  1629.9     .17       0  1745.4     .11       0  2208.1    .125       0
    2682     .15       0  2999.5     .11       0  4809.7     .06       0
  5262.6     .11       0  7065.4     .15       0  7549.2     .17       0
  8328.8     .17       0  8468.5     .15       0  8816.1     .11       0
 11026.7    .125       0 11207.4     .11       0
Bank Sta=4809.7,5262.6
XS Rating Curve= 0 ,0
Exp/Cntr=0.3,0.1

Type RM Length L Ch R = 1 ,179000  ,1334,1334,1334
BEGIN DESCRIPTION:
WFSJ Main 179.0
END DESCRIPTION:
XS GIS Cut Line= 3
       3870397.1     10061437.69      3863434.37     10057066.93
      3859382.16     10052987.88
#Sta/Elev= 30
 -3220.9  119.09 -1968.8  109.96  -184.2  104.18   938.1   95.87  1366.2   93.69
  1595.2   96.38  2263.3   80.09    3453   87.79  3855.7   91.99  4138.1   97.32
  4661.2   80.11  4998.1   63.44  5107.7   64.35  5143.1   78.79  5429.6   84.48
  5892.7   85.09    5928    72.5  5977.5   85.97  6189.6   87.14    6225   76.17
  6288.6   87.24  7434.4   88.03  7850.8   89.46  8167.3   92.14  8984.3   99.07
  9210.1  100.98  9477.2  103.25 10263.8  109.94 10510.2  109.05 10749.7  108.19
#Mann= 20 ,-1 , 0
 -3220.9     .17       0 -1968.8     .17       0  -184.2     .15       0
   938.1     .15       0  1366.2     .11       0  1595.2     .15       0
  2263.3     .11       0    3453     .15       0  3855.7     .11       0
  4661.2     .07       0  5143.1     .11       0  5429.6     .15       0
  7434.4     .15       0  7850.8     .17       0  8167.3     .11       0
  8984.3     .11       0  9210.1     .17       0  9477.2     .11       0
 10263.8     .11       0 10510.2    .125       0
Bank Sta=4661.2,5143.1
XS Rating Curve= 0 ,0
Exp/Cntr=0.3,0.1

Type RM Length L Ch R = 1 ,177666  ,1666,1666,1666
BEGIN DESCRIPTION:
WFSJ Main 178.0
END DESCRIPTION:
XS GIS Cut Line= 3
      3871399.67     10060565.28      3864837.17     10057049.65
      3860175.67     10052518.37
#Sta/Elev= 30
 -2655.6  106.91 -2579.7  106.86 -1640.5  106.25   -1548  106.19 -1444.6  106.12
     790   98.74  1852.4   92.19  1910.1   91.94  2206.6   92.26    3279   95.91
  3490.3   96.63  4153.7   91.35  4368.2   84.23  4929.1   90.57  4948.4   78.97
  4971.6   64.05  4998.1   62.78    5323  78.797  5473.7   87.51  5615.1   80.19
  5643.4   88.68    5700   83.12  6590.3   74.47  6640.7   67.64  6718.4   83.61
  7722.5   82.54  7807.4   90.26  9045.1  101.23 10736.7  105.24 11290.2  105.57
#Mann= 17 ,-1 , 0
 -2655.6     .17       0 -2579.7     .15       0 -1640.5     .17       0
   -1548     .15       0 -1444.6     .17       0     790     .15       0
  1852.4     .17       0  1910.1     .15       0  2206.6     .11       0
    3279     .17       0  3490.3     .11       0  4153.7     .11       0
  4948.4     .06       0    5323     .11       0  6590.3     .15       0
  9045.1     .17       0 10736.7     .11       0
Bank Sta=4948.4,5323
XS Rating Curve= 0 ,0
Exp/Cntr=0.3,0.1

Type RM Length L Ch R = 1 ,176000  ,1385,1385,1385
BEGIN DESCRIPTION:
WFSJ Main 176.0
END DESCRIPTION:
XS GIS Cut Line= 3
      3871881.46     10059627.79      3864805.66     10055293.44
       3860852.8     10051632.99
#Sta/Elev= 30
 -3297.8  104.32 -2553.5  104.81  -469.7   95.27  -166.1   95.98   442.3   94.36
   666.3   94.41  1509.7   86.19  1626.9   95.39  1995.3  105.91    2136    94.8
  2229.9  116.36  2273.7   95.02  2389.8  111.19  2432.4   92.49  2621.9   81.49
  3076.8   87.24  4591.8   76.52    4709   76.19  4998.1   62.49 5229.72   76.59
  6120.2   87.62  6319.3   88.43  6864.6   90.65  7340.5   92.59  7811.5    94.2
  8064.2   94.88  9082.4   97.63    9440    98.6 10034.9  107.19 10387.4  107.86
#Mann= 20 ,-1 , 0
 -3297.8     .15       0 -2553.5     .17       0  -469.7     .15       0
  -166.1     .17       0   442.3     .15       0   666.3     .17       0
  1626.9     .11       0  3076.8     .15       0  4591.8     .11       0
    4709     .07       0 5229.72     .15       0  6120.2     .11       0
  6319.3     .17       0  6864.6     .15       0  7340.5     .17       0
  7811.5     .15       0  8064.2     .15       0  9082.4     .17       0
    9440     .11       0 10034.9     .11       0
Bank Sta=4709,5229.72
XS Rating Curve= 0 ,0
Exp/Cntr=0.3,0.1

Type RM Length L Ch R = 1 ,174615  ,1615,1615,1615
BEGIN DESCRIPTION:
WFSJ Main 175.0
END DESCRIPTION:
XS GIS Cut Line= 3
      3872376.26     10059406.44      3865852.79     10054862.15
      3861752.05     10051204.03
#Sta/Elev= 30
 -2684.3  102.93   401.3   97.42   567.9   96.99  1740.6   97.92  1922.6    98.6
  2440.4  100.52  2705.7   95.89  2929.1   82.38  3346.6   84.64  3560.7   84.79
  3742.7   84.91  3932.1   85.04  4818.3   86.59 4905.73   74.46  4931.7   63.11
  4998.1   61.52 5353.5474.41957  5369.1   82.29  5846.5   82.53  5964.4   77.58
  6324.5   81.99  6717.7   83.22  7097.2    84.4  8204.7   89.39  8740.2   90.96
  9507.4    93.2  9781.8   91.03  9824.4   99.05 10097.5  102.17 10761.2  106.08
#Mann= 19 ,-1 , 0
 -2684.3     .17       0   401.3     .15       0   567.9     .17       0
  1740.6     .17       0  1922.6     .11       0  3346.6     .15       0
  3560.7     .11       0  3742.7     .17       0  3932.1     .15       0
 4905.73     .06       0 5353.54     .17       0  5846.5     .15       0
  6324.5     .17       0  6717.7     .15       0  7097.2     .15       0
  8204.7     .17       0  8740.2     .15       0  9507.4     .11       0
 10097.5     .17       0
Bank Sta=4905.73,5353.54
XS Rating Curve= 0 ,0
Exp/Cntr=0.3,0.1

Type RM Length L Ch R = 1 ,173000  ,2000,2000,2000
BEGIN DESCRIPTION:
WFSJ Main 173.0
END DESCRIPTION:
XS GIS Cut Line= 3
      3873274.64     10058364.74       3867204.5     10053902.34
      3862519.43     10050552.24
#Sta/Elev= 30
 -2533.9  102.34 -2249.7   96.85 -1547.2   94.66 -1173.4   93.49   462.6    92.9
   779.4   94.48  1407.9   94.34  1757.4   94.26  3479.7   87.35  3710.9   73.67
  3871.1   81.88  4142.8   84.57  4884.1   84.57 4909.09   75.35  4998.1   60.85
  5199.3   75.36  5436.4   86.67  5499.9   77.23  6389.6   87.91  6704.7   88.86
  6741.3   77.75  6882.2   87.14  7313.9   90.11  7521.5   77.57  7565.2   90.06
  8338.2    91.5    8690   92.05  9599.7   98.94 10546.2  106.48 10759.6  106.02
#Mann= 20 ,-1 , 0
 -2533.9     .11       0 -2249.7     .17       0 -1547.2     .15       0
 -1173.4     .17       0   462.6     .15       0   779.4     .17       0
  1407.9     .15       0  1757.4     .17       0  3479.7     .15       0
  3871.1     .11       0  4142.8     .15       0 4909.09     .09       0
  5199.3     .12       0  5436.4     .15       0  6389.6     .15       0
  6882.2     .11       0  8338.2     .17       0    8690     .15       0
  9599.7     .17       0 10546.2     .15       0
Bank Sta=4909.09,5199.3
XS Rating Curve= 0 ,0
Exp/Cntr=0.3,0.1

Type RM Length L Ch R = 1 ,171000  ,2000,2000,2000
BEGIN DESCRIPTION:
WFSJ Main 171.0
END DESCRIPTION:
XS GIS Cut Line= 4
       3874163.1      10057681.5      3873806.71     10057617.96
       3869024.6     10053742.64      3863021.34     10049025.41
#Sta/Elev= 30
       0  110.32     362   96.66  1312.3   92.29  5762.7   88.03    6303   81.69
    6359   62.58  6466.1    80.7  6501.2    60.5  6929.4   81.32  7335.2   88.32
  7583.8   77.99  7705.8   89.37  7904.6   77.98  8823.8   77.85  9030.7   87.25
 10041.2   91.19 10126.1   78.33 10312.3   89.57 10633.1   78.21 10689.2   93.69
 10974.7   94.81 11024.4   81.26   11095   80.55 11152.8   93.15   11273   90.74
 11316.4   78.14 11451.1   89.45 11508.9   77.78 11614.6   88.81 14150.6  109.15
#Mann= 3 , 0 , 0
       0    .125       0  6466.1     .06       0  6929.4    .125       0
#XS Ineff= 3 ,-1
 10041.2   10692   91.19 10974.7   12530   94.81  7705.8    9960   89.37
Permanent Ineff=
       F       F       F
Bank Sta=6466.1,6929.4
XS Rating Curve= 0 ,0
Exp/Cntr=0.3,0.1

Type RM Length L Ch R = 1 ,169000  ,2000,2000,2000
BEGIN DESCRIPTION:
WFSJ Main 169.0
END DESCRIPTION:
XS GIS Cut Line= 3
      3874711.29      10056376.9      3870140.21     10052312.51
      3864147.09     10047726.75
#Sta/Elev= 30
 -1116.7  125.71  1235.9   87.05  2418.5   78.31  3344.1   77.38  4151.7    81.5
  4287.3   80.12  4350.8   65.57  4641.8   76.77  4697.9   66.49  4998.1   59.61
  5138.7   76.78  5367.2   83.34  5608.3   74.84  5716.3   83.55  6097.9   78.87
  7063.4   84.47  7595.1   81.79  7908.2   87.41  7962.3   95.83  8084.7   81.37
  8348.6   81.69  8427.5    94.3  8873.7    88.4    9115   89.39  9834.7   89.17
 10303.1      89 10579.7   87.31 11202.5   93.38 11770.1    97.8 12546.3  103.84
#Mann= 20 ,-1 , 0
 -1116.7     .17       0  1235.9     .17       0  2418.5     .15       0
  3344.1     .15       0  4151.7     .17       0  4287.3     .11       0
  4641.8     .06       0  5138.7     .11       0  5716.3     .15       0
  6097.9     .11       0  7063.4     .11       0  7595.1     .17       0
  7908.2     .11       0  8873.7     .11       0    9115     .15       0
  9834.7     .11       0 10303.1     .15       0 10579.7     .17       0
 11202.5     .15       0 11770.1     .17       0
#XS Ineff= 1 ,-1
  7962.3   11670   95.83
Permanent Ineff=
       F
Bank Sta=4641.8,5138.7
XS Rating Curve= 0 ,0
Exp/Cntr=0.3,0.1
