HEC-RAS study WFSJ Main.prj: WFSJ Main Base Level Engineering

--- WFSJ Main.g02 (geometry) --- (continued)

Type RM Length L Ch R = 1 ,201926  ,1092,1092,1092
BEGIN DESCRIPTION:
WFSJ Main 202.0
END DESCRIPTION:
XS GIS Cut Line= 4
      3861250.82     10076007.56      3856276.84     10074106.51
      3855977.36     10073637.76      3847111.54     10072088.52
#Sta/Elev= 30
  -579.6  146.71   239.3  102.82   592.7  102.24   956.9  101.65  1231.5   101.2
  1577.9  101.98  3984.1  108.36  4091.2   87.54  4929.7   90.63  4998.1   75.76
 5465.91   90.87  5572.6  100.35  5834.1   83.71  6316.6   87.48  6567.4   95.28
  7064.8   89.04  7345.6   82.96  7412.6  100.55    7443   81.84  7548.2   88.48
  7762.3   89.53  7973.8   95.14  8217.8  110.37 10082.4  102.53 11787.9  113.68
 11820.6  125.72 11975.9  116.41 12595.5  117.95 14060.4  120.34 14301.7  118.38
#Mann= 18 ,-1 , 0
  -579.6     .12       0   239.3      .1       0   592.7     .12       0
   956.9     .12       0  1231.5     .05       0  1577.9     .05       0
  4929.7     .05       0 5465.91     .05       0  5572.6      .1       0
  6316.6     .05       0  6567.4      .1       0  7064.8     .05       0
  7548.2      .1       0  7762.3      .1       0  7973.8     .05       0
 11975.9     .12       0 12595.5     .05       0 14060.4      .1       0
#Block Obstruct= 3 ,-1
  8217.8   11245  110.37     -65  1835.6  112.94    1836  3984.1  108.36
Bank Sta=4929.7,5465.91
XS Rating Curve= 0 ,0
Exp/Cntr=0.3,0.1

Type RM Length L Ch R = 1 ,200834  ,834,834,834
BEGIN DESCRIPTION:
WFSJ Main 201.0
END DESCRIPTION:
XS GIS Cut Line= 4
       3862891.4     10074575.25      3856537.25     10073169.01
      3854308.11     10072459.15      3847344.56     10071997.13
#Sta/Elev= 30
 -1219.5   150.3  -580.9  103.25   902.3   99.53    1410   99.49  1601.6   99.48
  1735.2   99.47  2108.4   99.44  2128.4   99.44  2288.2   99.43  3842.5   99.32
  4898.6   90.45  4998.1   74.78 5102.29   91.22  5112.7   94.81  5676.1   99.23
  5987.5   91.24  6337.9   89.96  7371.7  100.32  8740.5   99.74  8780.6     114
  9281.7  115.73  9522.3  103.35 10263.9  113.12 10424.2   98.06 10835.1  110.99
 10915.3   98.75 12915.8   108.2 13184.3  118.28 14466.2   118.5 14606.7  118.42
#Mann= 18 ,-1 , 0
 -1219.5     .05       0   902.3     .12       0    1410      .1       0
  1601.6     .12       0  1735.2      .1       0  2108.4     .12       0
  2128.4      .1       0  2288.2     .12       0  3842.5      .1       0
  4898.6     .05       0  5112.7     .07       0  5676.1      .1       0
  5987.5     .05       0  6337.9      .1       0  7371.7     .05       0
 12915.8     .12       0 13184.3     .05       0 14466.2     .12       0
#Block Obstruct= 2 ,-1
  7340.4    9085  109.47  9281.7   13100  115.73
Bank Sta=4898.6,5102.29
XS Rating Curve= 0 ,0
Exp/Cntr=0.3,0.1

Type RM Length L Ch R = 1 ,200000  ,1000,1000,1000
BEGIN DESCRIPTION:
WFSJ Main 200.0
END DESCRIPTION:
XS GIS Cut Line= 4
      3863099.79     10073963.29      3856738.23     10072412.29
      3855026.84     10072049.22      3847474.75     10071814.84
#Sta/Elev= 30
 -1547.9  149.31  -578.4   99.71   -25.9  103.03   578.7    98.4   780.5   99.09
  1224.5   98.45  1752.2   98.88  2099.3  100.14  3149.5   98.91  3383.5   98.87
  4091.5   94.36  4619.9   98.82 4774.02  98.549 4801.97   91.37  4998.1   74.26
  5315.6   91.35  5327.5   91.53  5863.3   89.24  6042.8   89.05  6848.8   90.31
    7159   89.73  7288.7  109.43    7585   101.9  8299.2   95.12  9169.6  113.78
   11961   98.07 12611.3  118.39 12721.3  104.34   14288   119.4 14305.2  117.17
#Mann= 20 ,-1 , 0
 -1547.9     .05       0   -25.9     .12       0   578.7      .1       0
   780.5     .12       0  1224.5      .1       0  1752.2      .1       0
  2099.3     .12       0  3149.5     .12       0  3383.5      .1       0
  4091.5     .12       0  4619.9      .1       0 4774.02     .05       0
 4801.97     .03       0  5327.5     .05       0  5863.3     .05       0
  6042.8      .1       0  6848.8     .05       0    7159      .1       0
    7585     .05       0   14288     .12       0
#Block Obstruct= 2 ,-1
  7338.8    9066  109.18  9169.6   13127  113.78
Bank Sta=4801.97,5315.6
XS Rating Curve= 0 ,0
Exp/Cntr=0.3,0.1

Type RM Length L Ch R = 1 ,199000  ,1000,1000,1000
BEGIN DESCRIPTION:
WFSJ Main 199.0
END DESCRIPTION:
XS GIS Cut Line= 3
      3863568.51     10073142.97      3856608.15     10071429.79
      3849506.01      10070603.9
#Sta/Elev= 30
 -2168.1  140.79  -709.6  129.69  -381.3  125.78   174.8   98.07  3321.7   89.08
  3593.8   96.52  3635.3   88.47  4528.3    97.3  4725.1   99.78  4766.5   99.22
 4790.34   91.56  4835.5   75.47    4990   74.92  4998.1   74.42    5010   74.92
  5161.4   85.86  5312.4   78.69 5351.43   91.73  5372.8   99.27  5718.7   100.2
  6802.8   99.37  6953.1   94.54  7033.9     105  7758.8  101.85  8030.6  112.03
  8070.8   95.01    9138   95.47  9362.7  113.89  9962.7  104.19   12150  121.84
#Mann= 12 ,-1 , 0
 -2168.1     .05       0  -709.6     .12       0   174.8      .1       0
  4528.3     .12       0  4725.1     .05       0  4766.5     .05       0
    4990     .05       0    5010     .05       0  5372.8      .1       0
  5718.7     .05       0  6802.8      .1       0  6953.1     .05       0
#Block Obstruct= 1 ,-1
  8030.6   10640  112.03
Bank Sta=4790.34,5351.43
XS Rating Curve= 0 ,0
Exp/Cntr=0.3,0.1

Type RM Length L Ch R = 1 ,198000  ,1761,1761,1761
BEGIN DESCRIPTION:
WFSJ Main 198.0
END DESCRIPTION:
XS GIS Cut Line= 5
      3863724.79     10072791.41      3856913.52     10070661.55
      3855847.15     10069861.72      3854675.27     10068598.69
      3852762.04     10067817.78
#Sta/Elev= 30
 -2136.5  131.72 -1825.4  118.73   -12.8   125.2   410.7  106.51   819.4  104.88
   921.5  104.46  1149.3  103.53  4117.1    85.4  4673.5   91.28    4990   74.63
  4998.1   74.13    5010   74.63    5155   75.17  5182.1   91.02    5205   93.99
  5346.6   92.77  5382.1   82.34  5669.6  101.13  5816.4   86.67  6090.4   86.35
  6161.7  106.06  6207.1  109.43  7168.5  115.59  7301.2   116.7  7446.7  117.14
  7585.8  117.34  7731.6  118.32    8099  119.04  9668.8  118.27 10122.4     124
#Mann= 19 ,-1 , 0
 -2136.5     .05       0   410.7     .12       0   819.4      .1       0
   921.5     .12       0  1149.3      .1       0  4673.5     .05       0
    4990     .05       0    5010     .05       0    5205      .1       0
  5816.4     .05       0  6161.7     .12       0  6207.1     .05       0
  7168.5     .12       0  7301.2     .05       0  7446.7    .075       0
  7585.8     .05       0  7731.6    .075       0    8099     .05       0
  9668.8     .12       0
Bank Sta=4673.5,5182.1
XS Rating Curve= 0 ,0
Exp/Cntr=0.3,0.1

Type RM Length L Ch R = 1 ,196239  ,1239,1239,1239
BEGIN DESCRIPTION:
WFSJ Main 196.0
END DESCRIPTION:
XS GIS Cut Line= 3
      3864128.43     10072309.64      3858672.67     10069991.92
      3852904.43     10067570.04
#Sta/Elev= 30
 -1248.1     147   -1195  146.77  -888.9  147.64   110.6  115.05   474.6  108.91
  1735.8  103.73  2579.1  104.17  3904.5   94.88  4101.7   94.39  4852.7   94.17
    4928   89.92  4933.489.29115  4998.1   73.66  5216.5   77.75 5242.9289.42747
    5264   91.74  5287.8   80.28  5316.9   86.88  5499.5   88.09  5547.1   98.02
  5629.2   96.32  6888.5   98.85  7513.5  104.59  8076.3  116.52  8530.9  117.72
  8570.9   118.1  8771.6  119.81  8949.3  119.72  9889.7  115.36 10935.6  118.08
#Mann= 17 ,-1 , 0
 -1248.1     .12       0   -1195     .05       0  1735.8     .12       0
  2579.1      .1       0  3904.5     .12       0  4101.7      .1       0
  4852.7     .05       0    4928     .05       0    5264      .1       0
  5629.2      .1       0  6888.5     .12       0  7513.5     .05       0
  8530.9    .075       0  8570.9     .05       0  8771.6    .075       0
  8949.3     .05       0  9889.7     .12       0
Bank Sta=4933.4,5242.92
XS Rating Curve= 0 ,0
Exp/Cntr=0.3,0.1

Type RM Length L Ch R = 1 ,195000  ,1508,1508,1508
BEGIN DESCRIPTION:
WFSJ Main 195.0
END DESCRIPTION:
XS GIS Cut Line= 3
      3864948.68     10071307.02      3858877.01      10068844.6
      3852995.59     10067270.57
#Sta/Elev= 30
   -1552  136.13 -1250.8  137.78  -422.3  130.37   416.3   118.5   786.7  113.26
  1464.6  103.57  2176.4  104.93  2344.5   88.84  2398.4  101.51    2474   88.58
  2516.6   97.71  2551.5   88.67  2617.7  104.76  2830.1   110.4  2945.1  100.49
  3314.8  104.73  3598.3  101.84  4434.9   96.69  4713.6   81.16  4863.6   90.08
  4880.4    86.4  4998.1   72.67    5184   86.76  5273.5   96.58  6442.8   95.17
  6879.2   96.29  7436.3   97.71  7653.4   98.27  9778.5  110.16 11088.4  116.18
#Mann= 19 ,-1 , 0
   -1552     .05       0 -1250.8     .12       0  -422.3     .12       0
   416.3      .1       0   786.7     .05       0  1464.6     .05       0
  2617.7      .1       0  2945.1     .05       0  3314.8     .12       0
  3598.3      .1       0  4434.9     .12       0  4713.6      .1       0
  4863.6     .05       0  5273.5     .12       0  6442.8      .1       0
  6879.2     .05       0  7436.3     .12       0  7653.4     .05       0
  9778.5     .12       0
#Block Obstruct= 1 ,-1
     940  3165.1  108.68
Bank Sta=4880.4,5184
XS Rating Curve= 0 ,0
Exp/Cntr=0.3,0.1

Type RM Length L Ch R = 1 ,193492  ,1492,1492,1492
BEGIN DESCRIPTION:
WFSJ Main 193.0
END DESCRIPTION:
XS GIS Cut Line= 3
      3865722.57     10070226.73      3859993.42     10067791.84
      3853274.66     10066086.11
#Sta/Elev= 30
 -1505.4   144.8  -639.9  119.32  -287.5  117.57  1258.7  103.83  1575.1  102.51
  2306.9  105.81  2354.2  121.61  2422.2   87.88  2712.4   87.42  2900.3  108.74
  2965.2   99.31  3663.5  107.66  4738.5   95.29  4911.2   88.37  4921.5   83.44
  4998.1   70.73  5228.3   83.75  5406.4   83.79  5438.2    97.1  5716.2   96.39
    6452   96.01  6754.4   95.82    6956   98.46  8770.3   96.86  9759.6   98.97
 10067.8   98.71 10366.8    98.3 10478.3  108.83 10612.2  113.37 11651.6  114.72
#Mann= 18 ,-1 , 0
 -1505.4     .05       0  -639.9      .1       0  -287.5     .05       0
  1258.7      .1       0  1575.1     .05       0  4738.5      .1       0
  4911.2     .05       0  5406.4     .12       0  5716.2      .1       0
    6452     .05       0  6754.4     .12       0    6956      .1       0
  8770.3     .05       0  9759.6     .12       0 10067.8      .1       0
 10366.8     .12       0 10478.3     .05       0 10612.2     .12       0
#Block Obstruct= 2 ,-1
    2376  3663.5  107.66    -900  2354.2  121.61
Bank Sta=4921.5,5228.3
XS Rating Curve= 0 ,0
Exp/Cntr=0.3,0.1

Type RM Length L Ch R = 1 ,192000  ,2000,2000,2000
BEGIN DESCRIPTION:
WFSJ Main 192.0
END DESCRIPTION:
XS GIS Cut Line= 3
      3867024.66     10068338.71      3860434.33     10066448.65
      3853601.49     10065226.96
#Sta/Elev= 30
   -1856  137.15  -687.3  109.25     3.4  109.67   262.6  104.59  1238.2  101.84
  1647.3  101.38  2301.9  106.53  2755.9   94.71  2998.9   95.32    3680   95.62
  4714.7   93.36  4753.6   83.42  4809.1   73.11  4998.1   69.93    5067   71.83
 5094.0584.61525  5169.1   95.04  5219.9   87.43  6094.3   95.31  6506.7    94.7
  7203.4   99.64  7601.5      99  9424.2   95.56  9780.3   96.06 10217.9   96.84
 10467.9  114.64 10686.8  116.86 11283.9  114.67 11929.6  114.91 11941.2  114.91
#Mann= 18 ,-1 , 0
   -1856     .05       0     3.4      .1       0   262.6     .05       0
  1238.2      .1       0  1647.3     .05       0  2755.9     .05       0
  2998.9      .1       0    3680     .05       0  5169.1     .12       0
  6094.3      .1       0  6506.7     .05       0  7203.4     .12       0
  7601.5      .1       0  9424.2     .05       0  9780.3      .1       0
 10686.8     .05       0 11283.9     .05       0 11929.6      .1       0
Bank Sta=4753.6,5094.05
XS Rating Curve= 0 ,0
Exp/Cntr=0.3,0.1

Type RM Length L Ch R = 1 ,190000  ,2000,2000,2000
BEGIN DESCRIPTION:
WFSJ Main 190.0
END DESCRIPTION:
XS GIS Cut Line= 3
      3867805.92       10066646.      3859938.21     10064731.89
       3854055.9     10063312.67
#Sta/Elev= 30
 -3097.2  133.01 -2292.5  123.89 -1882.7  102.72  -737.1   99.44  -440.6   97.06
    23.5   96.16  1118.3   95.87  1625.1   94.29  2172.3   94.06  3158.6   95.22
  3536.2   94.48  4441.5   93.75  4763.7   94.57 4792.18   85.27    4990   70.16
  4998.1   69.66    5010   70.16    5045   75.01  5109.2   70.16  5156.8   85.71
  5407.6   97.01  6605.1   98.66    7257   99.08  7531.3   95.55  9050.1   97.52
  9444.3   98.02    9627  115.85 10258.5  113.66 10609.2  113.43 11051.1  113.78
#Mann= 20 ,-1 , 0
 -3097.2     .05       0 -1882.7     .12       0  -737.1      .1       0
  -440.6     .05       0    23.5      .1       0  1118.3      .1       0
  1625.1     .05       0  2172.3     .05       0  3158.6      .1       0
  3536.2      .1       0  4441.5     .05       0    4990     .05       0
    5010     .05       0    5045     .12       0  6605.1      .1       0
    7257     .05       0  7531.3      .1       0  9050.1      .1       0
 10258.5     .12       0 10609.2     .05       0
Bank Sta=4792.18,5156.8
XS Rating Curve= 0 ,0
Exp/Cntr=0.3,0.1

Type RM Length L Ch R = 1 ,188000  ,2000,2000,2000
BEGIN DESCRIPTION:
WFSJ Main 188.0
END DESCRIPTION:
XS GIS Cut Line= 3
      3868144.44     10065682.46       3860889.5     10063124.74
      3855111.68     10061047.43
#Sta/Elev= 30
 -2692.6  131.01 -2347.1  121.12 -1969.2  126.82 -1625.5  106.32   -1392   93.73
  2210.8   96.11  2832.3   94.14  4119.9   92.93  4158.4   92.66  4212.9   92.28
  4249.2   81.83  4578.9   81.18  4683.6   80.35  4998.1   68.59  5097.4   70.06
 5137.6381.74817  5175.2   92.74  6468.2   94.47  6723.3  100.67  6918.6   95.18
  7276.6    97.8  7307.7  105.37  7388.8   97.52  7864.4   99.98  7920.5   94.21
  8051.6  104.48  8124.9   96.31  8723.3  112.09 11109.1   115.2 11139.9  115.31
#Mann= 10 ,-1 , 0
 -2692.6     .05       0 -1969.2     .12       0 -1625.5     .05       0
  2210.8      .1       0  2832.3     .05       0  4119.9     .12       0
  4158.4     .05       0  4683.6     .03       0 5137.63     .05       0
 11109.1     .12       0
Bank Sta=4578.9,5137.63
XS Rating Curve= 0 ,0
Exp/Cntr=0.3,0.1

Type RM Length L Ch R = 1 ,186000  ,2000,2000,2000
BEGIN DESCRIPTION:
WFSJ Main 186.0
END DESCRIPTION:
XS GIS Cut Line= 3
      3868717.39     10064367.36      3861339.03     10061731.95
      3855475.21     10060669.45
#Sta/Elev= 30
 -2834.9  124.02 -1400.3  127.39  -669.2   93.51  1330.9    94.6  1473.1   92.77
  2156.7   94.98  2260.9   92.47  3160.3   94.02  3985.9   94.56  4293.8   93.47
  4485.7   93.16  4696.7   84.89 4709.97   78.36    4990   67.68  4998.1   67.18
    5010   67.68  5088.3   78.89  5141.8   89.45  5447.3   91.23  5853.6   87.64
  6773.1   88.94  7167.6  123.24  7318.3   111.6  8035.8  112.29  8135.4  112.01
 10167.4  114.09 10325.6  114.59 10524.7  113.92 10798.1  111.97 10959.3  112.07
#Mann= 20 ,-1 , 0
 -2834.9     .05       0  1330.9      .1       0  1473.1      .1       0
  2156.7      .1       0  2260.9     .05       0  3160.3      .1       0
  3985.9     .12       0  4293.8      .1       0  4485.7      .1       0
  4696.7     .05       0    4990     .05       0    5010     .05       0
  5447.3    .075       0  5853.6     .05       0  8035.8    .075       0
  8135.4     .05       0 10167.4     .12       0 10325.6     .05       0
 10524.7      .1       0 10798.1     .12       0
Bank Sta=4709.97,5088.3
XS Rating Curve= 0 ,0
Exp/Cntr=0.3,0.1

Type RM Length L Ch R = 1 ,184000  ,1109,1109,1109
BEGIN DESCRIPTION:
WFSJ Main 184.0
END DESCRIPTION:
XS GIS Cut Line= 3
       3868899.7      10063885.6      3860787.93     10059997.15
      3855917.93     10059380.38
#Sta/Elev= 30
 -3995.6  117.08  -345.8  100.13   -23.5   99.62      84   99.21   191.4   98.97
   254.2   98.83   298.8   98.73   728.5   95.43  1519.4   89.78  3192.5   76.06
  3226.2   92.56    3481  103.92  3843.9   91.63  4058.7   90.46  4313.3   77.62
  4375.7   89.17  4398.4   78.68  4501.1   72.51  4778.778.74182  4998.1   66.09
  5080.7   67.16 5097.55   79.22    5121   97.36  6038.3   87.43  6764.3    88.6
  6844.7   98.71  6874.9   88.68  6999.6   90.59  7036.2   105.3  9908.9  111.85
#Mann= 13 ,-1 , 0
 -3995.6     .05       0  -345.8      .1       0   -23.5     .12       0
      84      .1       0   191.4     .12       0   254.2      .1       0
   298.8     .12       0   728.5      .1       0  1519.4     .05       0
  3843.9     .12       0  4058.7     .05       0  4375.7     .03       0
    5121     .05       0
#XS Ineff= 1 ,-1
    5121    7150   97.36
Permanent Ineff=
       F
#Block Obstruct= 1 ,-1
   -1700    3481  103.92
Bank Sta=4778.7,5097.55
XS Rating Curve= 0 ,0
Exp/Cntr=0.3,0.1

Type RM Length L Ch R = 1 ,182891  ,1695,1695,1695
BEGIN DESCRIPTION:
WFSJ Main 183.0
END DESCRIPTION:
XS GIS Cut Line= 4
      3869094.97     10063677.25      3861764.25     10059679.86
      3860996.02     10058859.55      3856165.28     10058182.46
#Sta/Elev= 30
 -3768.4  114.57 -2431.2  124.04  -626.2  100.68  -327.4    98.1   302.9   96.73
   648.9   95.98  1060.8   95.08  1317.8   94.52  2218.7    91.3  2706.5   89.71
  2777.7  100.41  3324.4   94.44  3392.7   83.03  4172.2      90  4201.4   81.37
  4627.5   94.33  4733.5   76.43  4938.6   78.74  4998.1   65.65  5143.8   66.17
 5191.98   78.38  5214.6   91.03  5264.4   91.49  7089.7   96.31  7201.7   95.68
  7254.4   95.41  7974.9  101.83  8073.9  102.68  8432.5  105.74 10583.2  109.98
#Mann= 16 ,-1 , 0
 -3768.4     .05       0  -626.2     .12       0  -327.4      .1       0
   302.9     .12       0   648.9      .1       0  1060.8     .12       0
  1317.8      .1       0  2218.7     .05       0  4627.5     .03       0
  5264.4     .05       0  7089.7     .12       0  7201.7     .05       0
  7254.4     .12       0  7974.9     .05       0  8073.9     .12       0
  8432.5     .05       0
#XS Ineff= 1 ,-1
    6804    7575   97.49
Permanent Ineff=
       F
#Block Obstruct= 2 ,-1
    -815  2777.7  100.41  2777.8  4548.1   95.41
Bank Sta=4938.6,5191.98
XS Rating Curve= 0 ,0
Exp/Cntr=0.3,0.1

Type RM Length L Ch R = 1 ,181196  ,2196,2196,2196
BEGIN DESCRIPTION:
WFSJ Main 182.0
END DESCRIPTION:
XS GIS Cut Line= 4
      3869719.95     10062791.82      3863730.39     10058794.44
      3863144.46     10059067.88      3858418.79     10054009.12
#Sta/Elev= 30
 -3096.9  116.94 -2908.5  115.98 -2401.4   113.4 -1938.3  111.04  -549.1   99.22
  -100.5  107.69   515.8  103.42  1629.9   98.87  1745.4   97.96  2208.1   94.33
    2682   87.04  2999.5   91.13  4486.9   78.07  4526.2   90.19  4750.7   91.31
  4802.4   76.51  4809.7   80.37  4998.1   64.65  5262.6   80.81  5269.4   82.66
  7065.4   91.09  7257.7   91.33  7292.9   80.54  7549.2   91.26  8328.8   95.53
  8468.5   96.29  8816.1   98.19 11026.7   110.5 11207.4  110.38 11673.3  108.97
#Mann= 20 ,-1 , 0
 -3096.9     .12       0 -2908.5     .05       0 -2401.4     .12       0
 -1938.3      .1       0  -100.5     .12       0   515.8      .1       0
  1629.9     .12       0  1745.4     .05       0  2208.1    .075       0
    2682      .1       0  2999.5     .05       0  4802.4     .03       0
  5269.4     .05       0  7065.4      .1       0  7549.2     .12       0
  8328.8     .12       0  8468.5      .1       0  8816.1     .05       0
 11026.7    .075       0 11207.4     .05       0
Bank Sta=4809.7,5262.6
XS Rating Curve= 0 ,0
Exp/Cntr=0.3,0.1

Type RM Length L Ch R = 1 ,179000  ,1334,1334,1334
BEGIN DESCRIPTION:
WFSJ Main 179.0
END DESCRIPTION:
XS GIS Cut Line= 3
       3870397.1     10061437.69      3863434.37     10057066.93
      3859382.16     10052987.88
#Sta/Elev= 30
 -3220.9  119.09 -1968.8  109.96  -184.2  104.18   938.1   95.87  1366.2   93.69
  1595.2   96.38  2263.3   80.09    3453   87.79  3855.7   91.99  4661.2   80.11
    4990   63.94  4998.1   63.44    5010   63.94  5107.7   64.35  5143.1   78.79
  5429.6   84.48  5892.7   85.09    5928    72.5  5977.5   85.97    6225   76.17
  6288.6   87.24  7434.4   88.03  7850.8   89.46  8167.3   92.14  8984.3   99.07
  9210.1  100.98  9477.2  103.25 10263.8  109.94 10510.2  109.05 10749.7  108.19
#Mann= 20 ,-1 , 0
 -3220.9     .12       0 -1968.8     .12       0  -184.2      .1       0
   938.1      .1       0  1366.2     .05       0  1595.2      .1       0
  2263.3     .05       0    3453      .1       0  3855.7     .05       0
    4990     .05       0    5010     .05       0  5429.6      .1       0
  7434.4      .1       0  7850.8     .12       0  8167.3     .05       0
  8984.3     .05       0  9210.1     .12       0  9477.2     .05       0
 10263.8     .05       0 10510.2    .075       0
#Block Obstruct= 1 ,-1
    1540  4101.6   97.61
Bank Sta=4661.2,5143.1
XS Rating Curve= 0 ,0
Exp/Cntr=0.3,0.1

Type RM Length L Ch R = 1 ,177666  ,1666,1666,1666
BEGIN DESCRIPTION:
WFSJ Main 178.0
END DESCRIPTION:
XS GIS Cut Line= 3
      3871399.67     10060565.28      3864837.17     10057049.65
      3860175.67     10052518.37
#Sta/Elev= 30
 -2655.6  106.91 -2579.7  106.86 -1640.5  106.25   -1548  106.19 -1444.6  106.12
     790   98.74  1852.4   92.19  1910.1   91.94  2206.6   92.26    3279   95.91
  3490.3   96.63  4153.7   91.35  4368.2   84.23  4929.1   90.57  4943.3   83.42
  4948.4   78.97  4971.6   64.05  4998.1   62.78    5323  78.797  5473.7   87.51
  5615.1   80.19  5643.4   88.68  6590.3   74.47  6640.7   67.64  6718.4   83.61
  7722.5   82.54  7807.4   90.26  9045.1  101.23 10736.7  105.24 11290.2  105.57
#Mann= 17 ,-1 , 0
 -2655.6     .12       0 -2579.7      .1       0 -1640.5     .12       0
   -1548      .1       0 -1444.6     .12       0     790      .1       0
  1852.4     .12       0  1910.1      .1       0  2206.6     .05       0
    3279     .12       0  3490.3     .05       0  4153.7     .05       0
  4943.3     .03       0    5323     .05       0  6590.3      .1       0
  9045.1     .12       0 10736.7     .05       0
#Block Obstruct= 1 ,-1
     610  3722.3   98.52
Bank Sta=4948.4,5323
XS Rating Curve= 0 ,0
Exp/Cntr=0.3,0.1

Type RM Length L Ch R = 1 ,176000  ,1385,1385,1385
BEGIN DESCRIPTION:
WFSJ Main 176.0
END DESCRIPTION:
XS GIS Cut Line= 3
      3871881.46     10059627.79      3864805.66     10055293.44
       3860852.8     10051632.99
#Sta/Elev= 30
 -3297.8  104.32 -2553.5  104.81  -469.7   95.27  -166.1   95.98   442.3   94.36
   666.3   94.41  1626.9   95.39    2136    94.8  2229.9  116.36  2273.7   95.02
  2389.8  111.19  2432.4   92.49  2621.9   81.49  3076.8   87.24  4591.8   76.52
    4709   76.19    4990   62.99  4998.1   62.49    5010   62.99 5229.72   76.59
  6120.2   87.62  6319.3   88.43  6864.6   90.65  7340.5   92.59  7811.5    94.2
  8064.2   94.88  9082.4   97.63    9440    98.6 10034.9  107.19 10387.4  107.86
#Mann= 20 ,-1 , 0
 -3297.8      .1       0 -2553.5     .12       0  -469.7      .1       0
  -166.1     .12       0   442.3      .1       0   666.3     .12       0
  1626.9     .05       0  3076.8      .1       0  4591.8     .05       0
    4990     .07       0    5010      .1       0  6120.2     .05       0
  6319.3     .12       0  6864.6      .1       0  7340.5     .12       0
  7811.5      .1       0  8064.2      .1       0  9082.4     .12       0
    9440     .05       0 10034.9     .05       0
#Block Obstruct= 1 ,-1
 -3297.8  2389.8  111.19
Bank Sta=4709,5229.72
XS Rating Curve= 0 ,0
Exp/Cntr=0.3,0.1

Type RM Length L Ch R = 1 ,174615  ,1615,1615,1615
BEGIN DESCRIPTION:
WFSJ Main 175.0
END DESCRIPTION:
XS GIS Cut Line= 3
      3872376.26     10059406.44      3865852.79     10054862.15
      3861752.05     10051204.03
#Sta/Elev= 30
 -2684.3  102.93   401.3   97.42   567.9   96.99  1740.6   97.92  1922.6    98.6
  2440.4  100.52  2705.7   95.89  2929.1   82.38  3346.6   84.64  3560.7   84.79
  3742.7   84.91  3932.1   85.04    4882   81.92 4905.73   74.46  4931.7   63.11
  4998.1   61.52 5353.5474.41957  5369.1   82.29    5426   81.56  5846.5   82.53
  6324.5   81.99  6717.7   83.22  7097.2    84.4  8204.7   89.39  8740.2   90.96
  9507.4    93.2  9781.8   91.03  9824.4   99.05 10097.5  102.17 10761.2  106.08
#Mann= 19 ,-1 , 0
 -2684.3     .12       0   401.3      .1       0   567.9     .12       0
  1740.6     .12       0  1922.6     .05       0  3346.6      .1       0
  3560.7     .05       0  3742.7     .12       0  3932.1      .1       0
    4882     .03       0    5426     .12       0  5846.5      .1       0
  6324.5     .12       0  6717.7      .1       0  7097.2      .1       0
  8204.7     .12       0  8740.2      .1       0  9507.4     .05       0
 10097.5     .12       0
Bank Sta=4905.73,5353.54
XS Rating Curve= 0 ,0
Exp/Cntr=0.3,0.1

Type RM Length L Ch R = 1 ,173000  ,2000,2000,2000
BEGIN DESCRIPTION:
WFSJ Main 173.0
END DESCRIPTION:
XS GIS Cut Line= 3
      3873274.64     10058364.74       3867204.5     10053902.34
      3862519.43     10050552.24
#Sta/Elev= 30
 -2533.9  102.34 -2249.7   96.85 -1547.2   94.66 -1173.4   93.49   462.6    92.9
   779.4   94.48  1407.9   94.34  1757.4   94.26  3479.7   87.35  3710.9   73.67
  3871.1   81.88  4142.8   84.57  4891.4   82.87 4909.09   75.35  4998.1   60.85
  5199.3   75.36  5436.4   86.67  5499.9   77.23  6389.6   87.91  6704.7   88.86
  6741.3   77.75  6882.2   87.14  7313.9   90.11  7521.5   77.57  7565.2   90.06
  8338.2    91.5    8690   92.05  9599.7   98.94 10546.2  106.48 10759.6  106.02
#Mann= 19 ,-1 , 0
 -2533.9     .05       0 -2249.7     .12       0 -1547.2      .1       0
 -1173.4     .12       0   462.6      .1       0   779.4     .12       0
  1407.9      .1       0  1757.4     .12       0  3479.7      .1       0
  3871.1     .05       0  4142.8      .1       0  4891.4     .07       0
  5436.4      .1       0  6389.6      .1       0  6882.2     .05       0
  8338.2     .12       0    8690      .1       0  9599.7     .12       0
 10546.2      .1       0
Bank Sta=4909.09,5199.3
XS Rating Curve= 0 ,0
Exp/Cntr=0.3,0.1

Type RM Length L Ch R = 1 ,171000  ,2000,2000,2000
BEGIN DESCRIPTION:
WFSJ Main 171.0
END DESCRIPTION:
XS GIS Cut Line= 3
      3873860.62     10057661.64       3869024.6     10053742.64
      3863326.77     10049263.21
#Sta/Elev= 30
 -1224.6   97.96  -288.7   94.49      16   92.66  1877.1   92.02  4274.2   85.62
  4785.8   81.69  4841.8   62.58  4942.4   81.21 4955.37   77.47  4998.1      60
  5312.8   77.34  5406.5   80.61  5832.4   87.61  5893.8   85.05  6015.7   77.99
  6230.2   87.36  7599.4    81.2  8695.8   79.32  8915.4   79.65  9115.6   78.21
  9183.1   93.13  9457.2   94.81  9577.5   80.55  9755.5   90.74  9828.6   78.36
 10398.4   91.18 10718.1   93.69 11320.7   98.42   12124  104.73 12247.8   105.7
#Mann= 20 ,-1 , 0
 -1224.6      .1       0  -288.7      .1       0      16     .12       0
  1877.1      .1       0  4274.2     .05       0  4942.4     .03       0
  5406.5     .05       0  5832.4     .12       0  5893.8      .1       0
  6015.7     .05       0  6230.2     .05       0  7599.4     .05       0
  8695.8      .1       0  8915.4      .1       0  9183.1     .05       0
  9828.6      .1       0 10398.4      .1       0 10718.1      .1       0
 11320.7     .12       0   12124      .1       0
#XS Ineff= 2 ,-1
  8794.8    9457   89.57  9457.2   10870   94.81
Permanent Ineff=
       F       F
Bank Sta=4955.37,5312.8
XS Rating Curve= 0 ,0
Exp/Cntr=0.3,0.1

Type RM Length L Ch R = 1 ,169000  ,2000,2000,2000
BEGIN DESCRIPTION:
WFSJ Main 169.0
END DESCRIPTION:
XS GIS Cut Line= 3
      3874711.29      10056376.9      3870140.21     10052312.51
      3864147.09     10047726.75
#Sta/Elev= 30
 -1116.7  125.71  1235.9   87.05  2418.5   78.31  3344.1   77.38  4151.7    81.5
  4287.3   80.12  4350.8   65.57  4641.8   76.77  4697.9   66.49  4998.1   59.61
  5138.7   76.78  5367.2   83.34  5608.3   74.84  5716.3   83.55  6097.9   78.87
  7063.4   84.47  7595.1   81.79  7908.2   87.41  7962.3   95.83  8084.7   81.37
  8348.6   81.69  8427.5    94.3  8873.7    88.4    9115   89.39  9834.7   89.17
 10303.1      89 10579.7   87.31 11202.5   93.38 11770.1    97.8 12546.3  103.84
#Mann= 20 ,-1 , 0
 -1116.7     .12       0  1235.9     .12       0  2418.5      .1       0
  3344.1      .1       0  4151.7     .12       0  4287.3     .05       0
  4641.8     .03       0  5138.7     .05       0  5716.3      .1       0
  6097.9     .05       0  7063.4     .05       0  7595.1     .12       0
  7908.2     .05       0  8873.7     .05       0    9115      .1       0
  9834.7     .05       0 10303.1      .1       0 10579.7     .12       0
 11202.5      .1       0 11770.1     .12       0
#XS Ineff= 1 ,-1
  7962.3   11670   95.83
Permanent Ineff=
       F
Bank Sta=4641.8,5138.7
XS Rating Curve= 0 ,0
Exp/Cntr=0.3,0.1

Type RM Length L Ch R = 1 ,167000  ,2497,2497,2497
BEGIN DESCRIPTION:
WFSJ Main 167.0
END DESCRIPTION:
XS GIS Cut Line= 3
      3875805.07     10055265.82      3872088.42     10051992.78
       3866075.3     10045774.81
#Sta/Elev= 30
    47.6  125.59    1227  110.77  1502.2  109.76  1671.2  123.87  1785.9  120.66
  2040.2  113.54  2957.9   85.72  3832.4   64.42  4406.4   62.55    4449   77.77
  4718.5   78.67  4739.4   69.52 4880.7380.77588 4891.76   75.99  4916.8   60.87
  4998.1   58.62  5715.8    76.1  5737.2   84.36  5942.2   82.73    6827   83.13
  9435.5   87.97 10666.2   84.17 10694.2   93.52 10815.1   87.06 11420.9    86.5
 11728.4   89.05 12467.5   95.18 13017.3   99.74 13552.5  103.23 13649.9  101.91
#Mann= 19 ,-1 , 0
    47.6     .12       0    1227      .1       0  1502.2     .12       0
  1785.9     .05       0  2040.2     .12       0  2957.9      .1       0
  4718.5     .05       0 4880.73     .03       0  5737.2     .05       0
  5942.2      .1       0    6827      .1       0  9435.5     .05       0
 10694.2      .1       0 10815.1     .05       0 11420.9      .1       0
 11728.4     .12       0 12467.5     .05       0 13017.3    .075       0
 13552.5     .05       0
#XS Ineff= 1 ,-1
  9082.1   12250   92.15
Permanent Ineff=
       F
Bank Sta=4891.76,5715.8
XS Rating Curve= 0 ,0
Exp/Cntr=0.3,0.1

Type RM Length L Ch R = 1 ,164503  ,1519,1519,1519
BEGIN DESCRIPTION:
WFSJ Main 165.0
END DESCRIPTION:
XS GIS Cut Line= 3
      3876603.69     10054536.66       3874173.1     10052127.77
      3866595.13     10045265.93
#Sta/Elev= 30
    1764     124  3241.5  120.58  3320.7  112.36  3511.6  118.96  3645.9  104.48
    3752  113.14  3970.2   94.24  4020.7  103.82  4374.3   89.01  4505.5   98.22
  4777.3   93.35  4819.7   77.36  4998.1   57.62    5393   63.76  5555.8   77.35
  5966.1   80.11  6204.2   82.28  8972.6   82.12    9389   80.88 10006.2   83.97
 10398.4   95.47 11218.1   88.75 11768.4   84.04 12316.5   84.92   13159   92.09
 13877.3   94.25 14050.9   98.79 14438.5  102.45 15265.9  103.59 15409.1  103.81
#Mann= 19 ,-1 , 0
    1764     .05       0  3241.5     .12       0  3970.2     .12       0
  4505.5     .05       0  4819.7     .03       0  5555.8     .05       0
  5966.1     .12       0  6204.2      .1       0  8972.6      .1       0
    9389      .1       0 10006.2     .12       0 11218.1      .1       0
 11768.4     .12       0 12316.5     .12       0   13159      .1       0
 13877.3     .12       0 14050.9     .05       0 14438.5    .075       0
 15265.9    .075       0
#XS Ineff= 1 ,-1
   10766   14050   94.99
Permanent Ineff=
       F
Bank Sta=4819.7,5555.8
XS Rating Curve= 0 ,0
Exp/Cntr=0.3,0.1

Type RM Length L Ch R = 1 ,162984  ,2092,2092,2092
BEGIN DESCRIPTION:
WFSJ Main 163.0
END DESCRIPTION:
XS GIS Cut Line= 4
      3878235.58     10053573.93      3875527.27     10051178.12
       3874360.6     10050803.12       3866861.7     10045033.14
#Sta/Elev= 30
   734.9  124.17  1161.6  120.05  1734.2   110.7  1854.3  104.38  2413.4  114.05
  2817.9   117.8  3455.5   88.18    3758   85.95  4350.8   79.64    4458   72.47
  4864.9   72.82  4998.1   56.92  5270.9   62.68  5316.6   74.91  5686.6   72.58
  5730.1    73.3  5750.9   81.52    5907    81.4  6210.5   79.18  8639.9   80.25
  9478.4   83.55  9845.4   86.17 11154.2   90.32 11569.7    89.9 12468.9   85.87
 12947.9   92.35 13903.4   98.14 14115.3  106.09 14923.7  102.81 15038.1  102.55
#Mann= 19 ,-1 , 0
   734.9     .05       0  1161.6     .12       0  1734.2     .12       0
  2413.4     .12       0    3758      .1       0  4350.8     .05       0
  4864.9     .03       0  5316.6     .05       0  5750.9      .1       0
    5907     .12       0  6210.5      .1       0  8639.9      .1       0
  9478.4     .12       0  9845.4     .12       0 11154.2      .1       0
 11569.7     .12       0 12947.9     .12       0 13903.4     .05       0
 14923.7     .05       0
Bank Sta=4864.9,5316.6
XS Rating Curve= 0 ,0
Exp/Cntr=0.3,0.1

Type RM Length L Ch R = 1 ,160892  ,1892,1892,1892
BEGIN DESCRIPTION:
WFSJ Main 161.0
END DESCRIPTION:
XS GIS Cut Line= 4
      3878979.17     10052477.53      3875417.85     10049111.07
      3874742.37     10048970.47       3867155.6      10044456.6
#Sta/Elev= 30
  -206.9  119.46    2463    91.7    4043   68.24  4686.6   83.54  4846.9   73.51
  4877.6   63.15  4998.1   61.59 5145.56   73.74  5912.6   81.72  5997.8   82.51
  6282.8   73.96  6408.2    81.9  7115.1   74.06    7306   86.31  7348.8    72.7
  7426.5   72.38  7970.1   74.87  8065.2   88.82  8321.7   84.94  8527.2   82.74
  8579.2   83.68  8732.7   86.46  9149.3      94  9624.6   92.97 10472.5   93.32
 11497.1   90.99   11658   93.09 13015.1   100.3 13949.2  103.59 14211.7  104.23
#Mann= 20 ,-1 , 0
  -206.9     .12       0    2463      .1       0  4686.6     .05       0
  4846.9     .03       0 5145.56     .05       0  5912.6      .1       0
  5997.8     .05       0  6282.8      .1       0  7426.5     .05       0
  8321.7     .12       0  8527.2      .1       0  8579.2     .05       0
  8732.7     .12       0  9149.3     .05       0  9624.6     .12       0
 10472.5      .1       0 11497.1     .05       0   11658      .1       0
 13015.1     .12       0 13949.2      .1       0
#XS Ineff= 2 ,-1
  8065.2    8930   88.82  9319.7   12860   97.09
Permanent Ineff=
       F       F
Bank Sta=4846.9,5145.56
XS Rating Curve= 0 ,0
Exp/Cntr=0.3,0.1

Type RM Length L Ch R = 1 ,159000  ,2000,2000,2000
BEGIN DESCRIPTION:
WFSJ Main 159.0
END DESCRIPTION:
XS GIS Cut Line= 3
      3879152.84     10051557.44      3875399.55     10047372.46
      3867625.45     10043415.49
#Sta/Elev= 30
  -621.5     120  -469.9  119.48   470.1  115.34    1503   91.25    1886   79.84
  2878.7    79.1  4357.4   76.52  4499.5   68.56  4775.3    75.5  4782.8   72.75
  4998.1   61.04  5166.5   62.71  5188.7   72.76  5293.6   76.44  5322.2    65.7
  5344.5   76.01  5881.4   77.24  6200.9   77.97  6697.4   79.11  6941.1   79.67
  7196.7   80.25  7418.5   92.89  7764.5   92.96  8078.3      94  8406.6   93.12
  8701.8   94.59  9952.9   93.29 12448.3    96.3 13599.7  101.33 13723.2  101.87
#Mann= 19 ,-1 , 0
  -621.5     .12       0  -469.9     .05       0   470.1     .12       0
    1503      .1       0  2878.7     .05       0  4775.3     .03       0
  5188.7     .05       0  5881.4     .12       0  6200.9     .05       0
  6697.4     .12       0  6941.1      .1       0  7196.7     .12       0
  7764.5     .05       0  8078.3     .12       0  8406.6      .1       0
  8701.8     .12       0  9952.9      .1       0 12448.3      .1       0
 13599.7     .12       0
#XS Ineff= 1 ,-1
  9286.8   12600   95.78
Permanent Ineff=
       F
Bank Sta=4782.8,5188.7
XS Rating Curve= 0 ,0
Exp/Cntr=0.3,0.1

Type RM Length L Ch R = 1 ,157000  ,2000,2000,2000
BEGIN DESCRIPTION:
WFSJ Main 157.0
END DESCRIPTION:
XS GIS Cut Line= 4
      3880038.25      10050099.1      3877297.09     10047268.69
      3874811.82     10045133.67       3867921.2     10043189.71
#Sta/Elev= 30
  1059.8  118.88  1207.7  118.66  2016.1  116.18  2515.5  115.17  3958.2  114.13
  4296.3   82.38  4417.9   73.17  4870.6   68.75  4884.7   60.95  4998.1   60.14
  5281.3   68.51  5496.4   74.02  5707.1    71.6  5983.7   83.62  6266.8   82.13
  6628.9   91.88  6896.7   87.04  7609.1   88.39  8201.3   86.96  8585.9   88.06
  8955.8   89.26  9854.2   91.77 10172.5    92.5 10550.5    92.7 10983.6   92.62
 11686.6   91.78 12200.3   92.21 12490.5   91.21 14309.9   90.93   15436  101.71
#Mann= 20 ,-1 , 0
  1059.8     .05       0  1207.7     .12       0  2016.1     .12       0
  2515.5     .12       0  4296.3     .05       0  4870.6     .03       0
  5281.3     .05       0  5496.4     .12       0  6896.7     .05       0
  7609.1     .12       0  8201.3     .05       0  8585.9     .12       0
  8955.8      .1       0  9854.2      .1       0 10172.5     .12       0
 10550.5      .1       0 10983.6      .1       0 11686.6      .1       0
 12200.3     .12       0 12490.5      .1       0
#XS Ineff= 1 ,-1
  6628.9    9960   91.88
Permanent Ineff=
       F
Bank Sta=4870.6,5281.3
XS Rating Curve= 0 ,0
Exp/Cntr=0.3,0.1

Type RM Length L Ch R = 1 ,155000  ,2000,2000,2000
BEGIN DESCRIPTION:
WFSJ Main 155.0
END DESCRIPTION:
XS GIS Cut Line= 3
      3881184.04     10048935.86      3878097.98     10045468.91
      3868093.82     10041019.24
#Sta/Elev= 30
   358.5  112.72  1374.5  113.82  2087.9  104.23  2335.1   95.57  2916.2  100.73
  3164.2   91.19    3773   81.19  4237.2   74.47  4275.8   74.22  4736.5   78.96
  4807.6   71.01  4828.5   67.13  4998.1   59.38  5151.3   66.58  5428.9   76.27
  5459.8   65.73  5527.3   63.84  5568.4    72.7  5870.7   82.35  7226.1   85.51
  7669.6   86.58  7981.2   87.33  8776.6   88.89 10059.2   89.35 11179.5   92.11
 11565.1   90.43 12853.2   93.78 14501.5   96.39 14901.8   97.03 15949.1   98.69
#Mann= 20 ,-1 , 0
   358.5      .1       0  1374.5     .05       0  2087.9      .1       0
  3164.2      .1       0    3773     .12       0  4237.2     .12       0
  4275.8     .05       0  4807.6     .03       0  5151.3     .05       0
  5870.7     .12       0  7226.1     .12       0  7669.6     .05       0
  7981.2      .1       0  8776.6      .1       0 10059.2     .05       0
 11179.5     .05       0 11565.1      .1       0 12853.2      .1       0
 14501.5     .12       0 14901.8     .12       0
Bank Sta=4828.5,5151.3
XS Rating Curve= 0 ,0
Exp/Cntr=0.3,0.1

Type RM Length L Ch R = 1 ,153000  ,2000,2000,2000
BEGIN DESCRIPTION:
WFSJ Main 153.0
END DESCRIPTION:
XS GIS Cut Line= 3
      3882104.19     10047147.68      3878660.37     10043558.69
      3868754.29      10039005.7
#Sta/Elev= 30
      26  113.94   622.7  109.43   990.8  106.65  1634.2    97.2  2277.2   77.78
  3508.5   76.44  4118.1   78.62  4427.3   80.16  4538.5   74.61  4717.3   74.66
 4803.64    65.5  4998.1   59.22    5421   65.02    5454   64.92    5498   71.74
  5747.1   80.95  6423.5   78.71  7262.4   86.76  7516.9   87.48  7639.4   88.76
  7667.9   94.48  7834.3   88.46  8359.4   90.91  8959.7   89.95 10133.2   90.65
 10785.7   92.27 13973.8   90.94   14697   93.31 14990.8   94.27 15902.3   97.26
#Mann= 19 ,-1 , 0
      26      .1       0   622.7      .1       0   990.8     .12       0
  1634.2      .1       0  3508.5     .12       0  4118.1     .12       0
  4538.5      .1       0  4802.2     .03       0    5454     .05       0
  5747.1     .12       0  7262.4     .12       0  7516.9     .05       0
  8359.4     .05       0  8959.7     .12       0 10133.2     .12       0
 10785.7      .1       0 13973.8     .12       0   14697     .05       0
 14990.8     .12       0
Bank Sta=4803.64,5421
XS Rating Curve= 0 ,0
Exp/Cntr=0.3,0.1

Type RM Length L Ch R = 1 ,151000  ,2259,2259,2259
BEGIN DESCRIPTION:
WFSJ Main 151.0
END DESCRIPTION:
XS GIS Cut Line= 3
      3882972.26     10045949.78      3879133.97     10042029.41
      3869222.54     10038623.49
#Sta/Elev= 30
  -486.5   110.5   -61.8  104.47   593.1   95.42  1241.6   87.67  2704.9      76
  2775.6   60.95  2902.9   79.15  3429.1   73.41  3823.3   71.43  4055.6   58.53
  4861.7   64.66  4998.1   58.03 5256.91   65.06  5270.8   76.53  5723.1    76.4
  5963.8    86.9  6841.6   80.57  7223.7  106.48  7291.5   89.26  7523.1      81
  8313.9    88.2  8725.8   89.23  8946.2   89.79  9975.3   90.03 10197.5   90.94
   10798   90.35 13372.4   96.51 15221.6   92.38 15431.2   92.23 15480.3    92.2
#Mann= 20 ,-1 , 0
  -486.5     .05       0   -61.8     .05       0   593.1      .1       0
  1241.6      .1       0  3429.1      .1       0  3823.3     .05       0
  4861.7     .03       0 5256.91     .05       0  5270.8      .1       0
  5723.1     .05       0  6841.6     .05       0  8313.9     .12       0
  8725.8      .1       0  8946.2     .12       0  9975.3      .1       0
 10197.5     .12       0   10798      .1       0 13372.4     .12       0
 15221.6      .1       0 15431.2     .12       0
#Block Obstruct= 2 ,-1
  7223.7   16000  106.48  5963.8    7223    86.9
Bank Sta=4861.7,5256.91
XS Rating Curve= 0 ,0
Exp/Cntr=0.3,0.1

Type RM Length L Ch R = 1 ,148741  ,1510,1510,1510
BEGIN DESCRIPTION:
WFSJ Main 149.0
END DESCRIPTION:
XS GIS Cut Line= 4
       3883892.4     10043241.45      3881531.29     10042477.56
      3879812.54     10041297.01      3870247.06     10038015.93
#Sta/Elev= 30
  2092.3  106.93  2884.8  103.88  3530.4   81.51  3852.2   75.22  4633.2   69.58
  4855.1   67.79  4860.5    63.4  4998.1   56.93    5121    61.9 5249.87  63.274
  6250.3   74.77  6292.2   62.91  6507.4   59.26    6588   76.62  6800.8   77.51
  7640.5   76.41  8048.5   80.61  8942.5   96.39  9224.9   81.03  9839.6    81.2
 10272.7   90.13 10505.4   89.79 10956.3   89.12 11730.7   87.97 12681.5    89.1
 12903.4   89.86 13788.5    92.9 14003.1   93.64 15799.7   95.17 16771.6   95.54
#Mann= 20 ,-1 , 0
  2092.3     .05       0  3530.4     .12       0  3852.2      .1       0
  4633.2     .05       0  4855.1     .03       0    5121     .05       0
  6800.8      .1       0  7640.5     .12       0  8048.5     .05       0
  9224.9     .05       0  9839.6     .05       0 10272.7     .05       0
 10505.4     .12       0 10956.3      .1       0 11730.7      .1       0
 12681.5     .12       0 12903.4      .1       0 13788.5     .12       0
 14003.1      .1       0 15799.7     .12       0
#Block Obstruct= 1 ,-1
  8942.5   16771   96.39
Bank Sta=4860.5,5249.87
XS Rating Curve= 0 ,0
Exp/Cntr=0.3,0.1

Type RM Length L Ch R = 1 ,147231  ,2448,2448,2448
BEGIN DESCRIPTION:
WFSJ Main 147.0
END DESCRIPTION:
XS GIS Cut Line= 3
      3884605.29     10041782.93      3883302.12     10041574.78
      3871862.87      10036506.1
#Sta/Elev= 30
  1919.2  106.82  2188.3  104.91  2372.3  100.13  2585.4  108.98  3043.1  102.61
  3276.4   79.62  3385.6   78.58  4081.6   72.69  4328.5   66.81  4443.2    65.6
    4524   56.88  4762.3   63.61  4998.1   56.38 5212.76   64.22  5237.4   70.88
    5336   63.12  5540.5   69.51  5716.8   68.76  6262.4   65.44  6979.7   75.43
  8091.7    77.6  8950.7   80.22  9198.7   82.19 11876.5   86.89 12456.7   87.09
 12949.6   87.39 13573.9   90.97 14022.5   89.63 14310.1   92.38 15750.8   95.72
#Mann= 20 ,-1 , 0
  1919.2     .12       0  2188.3     .12       0  2585.4     .12       0
  3385.6      .1       0  4081.6      .1       0  4328.5     .05       0
  4443.2     .03       0  5237.4     .05       0  5540.5     .12       0
  5716.8      .1       0  6979.7     .12       0  8091.7      .1       0
  8950.7     .05       0  9198.7      .1       0 11876.5      .1       0
 12456.7     .12       0 12949.6     .12       0 13573.9     .12       0
 14022.5      .1       0 14310.1     .12       0
Bank Sta=4762.3,5212.76
XS Rating Curve= 0 ,0
Exp/Cntr=0.3,0.1

Type RM Length L Ch R = 1 ,144783  ,1915,1915,1915
BEGIN DESCRIPTION:
WFSJ Main 145.0
END DESCRIPTION:
XS GIS Cut Line= 3
      3885192.46     10039614.88      3882850.74     10039300.48
      3873059.03     10035290.05
#Sta/Elev= 30
  2967.7  107.46  3324.6   106.5  3527.3  103.88  3674.9   89.29  4092.3   71.99
  4606.9   74.78  4778.4   60.85  4859.1   65.61  4889.4   57.45  4998.1    55.4
 5252.5564.92963  5278.2   64.75  5452.7    59.2    5571   71.04  5852.3   70.91
  6400.8   71.88  6750.9   72.83  7992.4    75.8  8362.6   75.63  9108.1   75.87
 11048.2   80.94 11583.6   82.09 11938.5   82.75 12945.5   85.17 13241.2   84.42
 13722.6   85.74 14654.8   84.39 14999.2   96.89 15288.7   92.25 15911.6  100.38
#Mann= 20 ,-1 , 0
  2967.7     .12       0  3324.6     .05       0  3674.9      .1       0
  4859.1     .07       0 5252.55      .1       0  5278.2      .1       0
    5571     .12       0  5852.3      .1       0  6400.8      .1       0
  6750.9     .12       0  7992.4      .1       0  8362.6     .12       0
  9108.1      .1       0 11048.2     .12       0 11583.6     .05       0
 11938.5      .1       0 12945.5      .1       0 13241.2      .1       0
 13722.6     .05       0 15288.7     .12       0
Bank Sta=4859.1,5252.55
XS Rating Curve= 0 ,0
Exp/Cntr=0.3,0.1

Type RM Length L Ch R = 1 ,142868  ,2211,2211,2211
BEGIN DESCRIPTION:
WFSJ Main 143.0
END DESCRIPTION:
XS GIS Cut Line= 4
      3886165.18     10037830.17      3881479.21     10037321.31
      3878649.35     10035463.67      3874257.02     10033727.58
#Sta/Elev= 30
  1955.1  107.53    2450  106.04  2777.2   97.36  2941.2    84.9  3734.3   72.03
  4195.5   72.77  4235.8   60.45  4406.8   64.96  4477.2   57.06  4688.4   69.02
 4856.48   65.13  4998.1   54.78  5191.3   56.33  5251.7   65.04  5573.6   58.49
  5623.9   71.83  6112.2   72.94  6320.1   71.98  6818.2   76.81  7395.2   75.91
    7624   74.98  9700.3   82.47 10954.1   83.35   11276   83.78 11646.2      85
 12063.3   82.41 12277.9   84.73 13281.3   83.34 14092.2   94.81 14776.7   95.54
#Mann= 20 ,-1 , 0
  1955.1     .12       0    2450     .05       0  2941.2     .12       0
  3734.3     .05       0 4856.48     .03       0  5251.7     .05       0
  5623.9      .1       0  6112.2     .12       0  6320.1      .1       0
  6818.2     .12       0  7395.2     .05       0    7624      .1       0
  9700.3     .05       0 10954.1     .12       0   11276     .05       0
 11646.2     .12       0 12063.3      .1       0 12277.9     .05       0
 13281.3     .05       0 14092.2     .05       0
Bank Sta=4856.48,5251.7
XS Rating Curve= 0 ,0
Exp/Cntr=0.3,0.1

Type RM Length L Ch R = 1 ,140657  ,1787,1787,1787
BEGIN DESCRIPTION:
WFSJ Main 141.0
END DESCRIPTION:
XS GIS Cut Line= 3
      3890894.78     10036015.93      3883655.16     10035898.74
       3875777.6     10032344.07
#Sta/Elev= 30
 -2601.6  100.11 -1372.1  102.59 -1034.5   73.81    -609   74.71   113.7    68.3
   501.4   74.27  3686.2   73.26  4156.2   55.86  4366.2   67.06    4747   62.09
  4778.6   58.94  4998.1   53.92 5110.1161.62156  5118.7   65.78  5329.4   70.68
  6303.9   62.02  6897.5   74.67  7142.8   75.43  7538.1   73.07  7846.9   80.32
  8236.3   82.41  8509.6   82.62  9225.2   82.52 10098.5   81.04 11266.9      89
 11853.1   97.12 12491.3   96.35 12810.4   94.53 13165.7   94.23 13281.4   95.02
#Mann= 20 ,-1 , 0
 -2601.6     .05       0    -609      .1       0   113.7     .05       0
   501.4     .05       0  4778.6     .03       0  5118.7     .05       0
  5329.4      .1       0  6897.5     .05       0  7142.8      .1       0
  7538.1     .12       0  7846.9     .05       0  8236.3     .12       0
  8509.6      .1       0  9225.2     .05       0 10098.5     .12       0
 11266.9     .05       0 11853.1     .05       0 12491.3     .05       0
 12810.4      .1       0 13165.7     .05       0
#XS Ineff= 1 ,-1
   -1125    2286   75.97
Permanent Ineff=
       F
Bank Sta=4747,5110.11
XS Rating Curve= 0 ,0
Exp/Cntr=0.3,0.1

Type RM Length L Ch R = 1 ,138870  ,3207,3207,3207
BEGIN DESCRIPTION:
WFSJ Main 139.0
END DESCRIPTION:
XS GIS Cut Line= 3
      3890881.74     10035755.52      3883381.73     10034531.55
      3877602.85     10031616.08
#Sta/Elev= 30
 -1714.9  101.88  -539.7   99.45    43.6   74.28   281.2    72.9   330.6   60.42
  1227.4   58.64  1338.9   73.91  1622.6    59.7  3424.4   71.61  3629.7   70.62
  4492.7   73.48  4621.5   58.71  4824.4   59.58  4998.1    53.3 5137.0359.23381
  5240.6    62.5  5884.5   65.29  6057.1   55.56    6124   68.57  7429.8    76.4
  7674.7   75.75  7883.7   72.22  8523.7   77.98  8759.1   78.47 10384.4   81.32
 10722.5   83.79 11081.5   84.42 11257.6   82.74 11468.3   85.98   12357   97.07
#Mann= 20 ,-1 , 0
 -1714.9     .05       0    43.6      .1       0   281.2     .05       0
  3424.4      .1       0  3629.7     .05       0  4621.5     .05       0
  4824.4     .03       0 5137.03     .05       0  5240.6     .12       0
  5884.5      .1       0  7429.8     .05       0  7674.7     .12       0
  7883.7      .1       0  8523.7     .12       0  8759.1      .1       0
 10384.4     .05       0 10722.5     .12       0 11081.5     .05       0
 11257.6     .12       0 11468.3     .05       0
#Block Obstruct= 1 ,-1
    -230  2797.9   74.92
Bank Sta=4824.4,5137.03
XS Rating Curve= 0 ,0
Exp/Cntr=0.3,0.1

Type RM Length L Ch R = 1 ,135663  ,2663,2663,2663
BEGIN DESCRIPTION:
WFSJ Main 137.0
END DESCRIPTION:
XS GIS Cut Line= 3
      3891116.08     10035416.96      3882965.06     10032109.68
       3877731.8     10029662.28
#Sta/Elev= 30
 -3394.6   92.46 -1712.1    89.9 -1506.7   77.24 -1163.7   71.55  -452.1   59.35
  -163.5   67.62   -10.7   59.94  1092.9   79.25  1582.7   68.96  1636.3   84.37
  3578.3   58.21  3823.2   85.62  3918.5   63.61  4162.3   52.41  4877.5   58.11
    4998   49.55  5075.1   58.64  5125.4   79.99  5320.3      80    5566    78.7
  5716.9   79.38  6594.1   76.57  6724.3   78.46  6833.7   80.05  7677.5   80.63
  8542.9   83.04  9121.3   77.05  9626.8   78.12  9826.6   86.16 11179.1   94.81
#Mann= 20 ,-1 , 0
 -3394.6     .05       0 -1506.7      .1       0 -1163.7     .05       0
  -452.1     .05       0  -163.5      .1       0   -10.7     .05       0
  4877.5     .03       0  5075.1     .05       0  5125.4     .05       0
  5320.3     .12       0    5566     .12       0  5716.9     .05       0
  6594.1     .12       0  6724.3     .05       0  6833.7     .12       0
  7677.5      .1       0  8542.9      .1       0  9121.3     .05       0
  9626.8    .075       0  9826.6     .05       0
#Block Obstruct= 1 ,-1
   -1750  3823.2   85.62
Bank Sta=4877.5,5075.1
XS Rating Curve= 0 ,0
Exp/Cntr=0.3,0.1
