HEC-RAS study WOODSONS GULLY.prj: WOODSONS GULLY Base Level Engineering

--- WOODSONS GULLY.g10 (geometry) --- (continued)

Type RM Length L Ch R = 1 ,40900   ,402,402,402
BEGIN DESCRIPTION:
WOODSONS GULLY 80.0
END DESCRIPTION:
XS GIS Cut Line= 3
      3868083.95     10042918.54      3868623.86     10041879.51
      3868023.42     10041115.31
#Sta/Elev= 30
  3825.7  100.76  4048.2   98.54  4124.2   99.21  4240.4   98.85    4279   98.03
  4317.6   98.61    4330   97.87  4352.5   98.27  4693.5   92.39  4859.2   91.81
  4881.3   92.67    4909   92.15  4925.5   92.73  4975.4   92.14  5003.4   91.18
  5011.4   91.18  5020.4   92.25  5198.5   91.92    5221   92.72  5291.6    92.5
  5299.7   93.15  5354.9    93.5  5490.6   95.86  5527.4   95.96  5533.8   95.38
  5583.5   97.17  5605.1   96.66  5783.1   98.38  5883.5   97.98  5968.5  101.41
#Mann= 4 ,-1 , 0
  3825.7      .1       0  4975.4     .03       0  5020.4      .1       0
  5354.9     .12       0
Bank Sta=4975.4,5020.4
XS Rating Curve= 0 ,0
Exp/Cntr=0.3,0.1

Type RM Length L Ch R = 1 ,40498   ,498,498,498
BEGIN DESCRIPTION:
WOODSONS GULLY 79.0
END DESCRIPTION:
XS GIS Cut Line= 3
      3868079.58     10042957.65      3868808.24     10042044.55
      3869217.87     10041561.05
#Sta/Elev= 30
  3831.8  100.98  4006.5   98.81  4112.4   99.33  4170.1   98.32  4269.4   98.97
  4368.6    97.3    4383   97.75  4390.3   96.96  4432.7   97.29  4589.6   94.31
  4682.5    93.3  4703.3   94.14  4717.7   92.93    4825   91.72  4874.6    92.2
  4891.4   91.08  4909.9   92.16  5044.3   91.71  5080.6   91.93  5087.1    92.7
  5136.5   91.66  5201.2    92.8    5208   92.14  5257.4   93.63  5300.3   93.36
  5392.5   95.45  5505.7   96.31  5577.1   98.52  5607.3   97.53  5633.7   97.85
#Mann= 4 ,-1 , 0
  3831.8      .1       0  4874.6     .03       0  4909.9      .1       0
  5607.3     .12       0
Bank Sta=4874.6,4909.9
XS Rating Curve= 0 ,0
Exp/Cntr=0.3,0.1

Type RM Length L Ch R = 1 ,40000   ,381,381,381
BEGIN DESCRIPTION:
WOODSONS GULLY 78.0
END DESCRIPTION:
XS GIS Cut Line= 3
      3868096.91     10042994.12       3868995.8     10042344.43
       3869311.5     10041584.39
#Sta/Elev= 30
  3890.9  100.99    4002   99.08  4064.8   99.88  4108.7   98.76  4401.9   97.87
  4431.3   96.51  4552.8   96.29  4595.4   94.83  4825.1   93.41  4931.8   91.67
  5013.7   92.07  5021.3   90.72  5048.4   92.04  5101.5   92.67  5125.4   91.74
  5155.2   92.79  5178.5   91.57  5255.6   92.47  5356.4   91.82  5371.8      92
  5393.5   93.82  5481.3   94.37  5510.4    95.4  5515.8   94.59  5622.1   95.64
  5693.7   97.91  5741.3   97.68  5755.4   97.71  5783.3   97.24    5823   99.05
#Mann= 6 ,-1 , 0
  3890.9      .1       0  5013.7     .03       0  5048.4      .1       0
  5481.3     .12       0  5741.3      .1       0  5755.4     .12       0
Bank Sta=5013.7,5048.4
XS Rating Curve= 0 ,0
Exp/Cntr=0.3,0.1

Type RM Length L Ch R = 1 ,39619   ,418,418,418
BEGIN DESCRIPTION:
WOODSONS GULLY 77.0
END DESCRIPTION:
XS GIS Cut Line= 3
      3868207.48     10043127.77      3869302.97     10042343.05
      3869322.07     10041589.54
#Sta/Elev= 30
    3659  101.16    3907   97.59  4065.4   97.55  4087.5   96.44  4280.4    94.3
  4416.7   93.89  4446.2   92.93  4532.2   96.18  4538.3    95.3  4559.2   96.45
  4588.7   95.33  4645.2   96.04  4659.9   94.73  4717.3   94.54  4760.7   93.24
  4790.1   91.23    4811   91.45  4842.6   90.51  4889.5   91.57  5128.6   91.23
  5298.6   92.43  5338.6   91.54  5403.4   92.91  5458.7   94.44  5528.7   94.74
  5568.7   96.75  5608.7   95.76  5648.7   98.02  5688.7   96.81  5760.3   99.02
#Mann= 4 ,-1 , 0
    3659      .1       0    4811     .03       0  4889.5      .1       0
  5403.4     .12       0
Bank Sta=4811,4889.5
XS Rating Curve= 0 ,0
Exp/Cntr=0.3,0.1

Type RM Length L Ch R = 1 ,39201   ,423,423,423
BEGIN DESCRIPTION:
Mapping XS 26df1587
END DESCRIPTION:
XS GIS Cut Line= 3
      3868218.81     10043160.67      3869559.93     10042418.49
      3869972.24     10041849.94
#Sta/Elev= 30
  3352.7  101.04  3593.3    97.4  3793.8   95.61  3837.3   95.93  3853.3   95.15
  3875.1   95.07  3880.8   95.92  3918.6   93.94  3962.1   93.87  3968.8   94.55
  4021.6   92.84  4071.6   93.38  4152.2   92.62  4243.1   94.14  4374.3   92.65
  4403.1   91.21  4417.9      92  4433.9   91.13  4483.1   91.98  4596.5   91.39
  4824.4   92.04  4851.9   91.31  4856.2   90.42  4895.6   91.96  4931.7   91.13
  5167.8   91.73  5211.9   90.97  5318.6   93.47  5469.3   98.52  5587.8    99.7
#Mann= 3 , 0 , 0
  3352.7      .1       0  4824.4     .03       0  4895.6      .1       0
Bank Sta=4824.4,4895.6
XS Rating Curve= 0 ,0
Exp/Cntr=0.3,0.1

Type RM Length L Ch R = 1 ,38778   ,330,330,330
BEGIN DESCRIPTION:
WOODSONS GULLY 76.0
END DESCRIPTION:
XS GIS Cut Line= 3
      3868222.79     10043194.94      3869910.26     10042374.65
      3870017.86     10041911.05
#Sta/Elev= 30
  3203.8  100.96  3247.7  100.99  3315.3   98.74  3442.9   96.97  3665.3   95.75
    3755   93.83  3839.7   93.13  3854.3   93.87    3975    91.9  4265.7   91.41
  4354.7   92.29  4476.8   91.36  4521.5   92.62  4578.1   91.54  4654.9   92.34
  4707.9   91.51  4798.1   92.18  4832.8   90.98  5034.8   91.43  5039.7   90.44
 5103.07  91.474  5175.5   91.74  5180.6   92.91  5228.4   93.66  5278.8   92.88
  5371.2   95.72    5399    97.8  5412.3   96.57  5504.7    98.9    5556   99.02
#Mann= 3 , 0 , 0
  3203.8      .1       0  5034.8     .03       0 5103.07      .1       0
Bank Sta=5034.8,5103.07
XS Rating Curve= 0 ,0
Exp/Cntr=0.3,0.1

Type RM Length L Ch R = 1 ,38448   ,480,480,480
BEGIN DESCRIPTION:
WOODSONS GULLY 75.0
END DESCRIPTION:
XS GIS Cut Line= 3
      3867810.86     10043990.54      3870002.71     10042679.77
       3870200.2     10042161.08
#Sta/Elev= 30
  2293.2  102.78    2313  103.34  2335.7  101.66  2384.3  100.91    2501  101.46
  2532.1  100.51  2590.5  101.13  2814.2   99.63  2823.9   98.78  3078.7   95.46
  3115.7   96.27  3128.6   94.83  3268.4   93.93  3275.2   92.96  3296.6   93.43
  3333.5   92.25    3851   91.36  3860.3   90.24 3877.31  91.343  4606.4   91.54
  4674.4   91.61  4756.1   91.91    4859   91.82  4879.4   93.21  4934.2   90.97
  5123.5   91.14    5274    97.1  5353.7   98.75  5391.4   98.25  5402.1   99.17
#Mann= 7 ,-1 , 0
  2293.2      .1       0    3851     .03       0 3877.31      .1       0
  4606.4     .12       0  4674.4      .1       0  4756.1     .12       0
    4859      .1       0
Bank Sta=3851,3877.31
XS Rating Curve= 0 ,0
Exp/Cntr=0.3,0.1

Type RM Length L Ch R = 1 ,37968   ,384,384,384
BEGIN DESCRIPTION:
WOODSONS GULLY 74.0
END DESCRIPTION:
XS GIS Cut Line= 3
       3868179.8     10044645.91      3870342.12     10042804.77
      3870536.57     10042118.98
#Sta/Elev= 30
  1910.8  102.54  1955.5  102.49  1962.1  101.25  2132.3   96.65  2146.6   97.37
  2168.6   95.31  2232.3   93.75  2275.1   94.74  2281.7   95.94  2324.5   92.71
  2438.9   91.45  2659.8    91.4    3261   90.64    3516   90.89  3565.4   92.26
  3622.5   90.94  3799.5   91.06  3809.2   89.92  3821.2   91.02    4098   90.81
  4147.4   92.33  4268.2   91.01  4338.4   92.57  4381.3   91.35  4660.5   91.84
  4796.9   91.44    5108   90.89  5253.5   97.35  5380.1  100.86  5463.6  100.88
#Mann= 7 ,-1 , 0
  1910.8      .1       0  2438.9     .12       0  2659.8      .1       0
  3565.4     .03       0  4147.4      .1       0  4660.5     .12       0
  4796.9      .1       0
Bank Sta=3565.4,4147.4
XS Rating Curve= 0 ,0
Exp/Cntr=0.3,0.1

Type RM Length L Ch R = 1 ,37584   ,647,647,647
BEGIN DESCRIPTION:
WOODSONS GULLY 73.0
END DESCRIPTION:
XS GIS Cut Line= 3
      3871698.01     10043910.37      3870738.82     10042584.43
      3870630.31     10042159.06
#Sta/Elev= 30
  3262.8   96.16  3272.5   96.11  3334.8   93.92  3361.9   95.32  3391.3   91.99
  3420.7   92.56  3434.7   91.06  3462.4   93.44  3484.1   91.41  3524.6   90.87
  3692.9   91.16  3706.3   92.76  3728.5   92.54  3799.7   95.21  3900.2   93.07
  3928.4   91.12  3965.2   91.01  3967.1   89.63    4237   93.17  4243.6   92.25
    4273   92.09  4344.2   93.49  4385.9   91.25  4440.4   90.76  4515.9   92.44
  4601.7   92.84  4637.3   90.89  5026.6   90.68  5294.9  100.19  5338.3  100.76
#Mann= 6 ,-1 , 0
  3262.8      .1       0  3272.5     .12       0  3524.6      .1       0
  3900.2     .03       0    4237     .12       0  4440.4      .1       0
Bank Sta=3900.2,4237
XS Rating Curve= 0 ,0
Exp/Cntr=0.3,0.1

Type RM Length L Ch R = 1 ,36937   ,584,584,584
BEGIN DESCRIPTION:
WOODSONS GULLY 72.0
END DESCRIPTION:
XS GIS Cut Line= 3
      3871775.29     10043928.19      3871130.75     10042619.58
       3871098.2     10042031.51
#Sta/Elev= 30
  3508.5   95.21  3544.6   95.15  3669.7      93  3676.6   94.33  3775.6   91.79
  3832.5   91.16  3852.1   92.37  3871.8   92.42  3899.9   90.24  3922.3   91.48
  3989.7   90.05  4229.9   91.56  4252.2      90  4296.7   90.37  4299.5   89.08
  4363.6   91.88  4389.9   93.59    4439   94.47  4579.7   91.48  4653.4   90.58
  4686.1   92.98    4731   90.54    4804   90.56  4909.8   93.67  4938.8   90.78
  5015.8   90.14  5105.5    92.3  5226.1   92.26  5353.8   96.01  5556.2    99.3
#Mann= 10 ,-1 , 0
  3508.5      .1       0  3544.6     .12       0  3676.6     .05       0
  3775.6     .12       0  3852.1      .1       0  4229.9     .03       0
  4363.6      .1       0  4389.9     .12       0  4579.7      .1       0
  5353.8     .12       0
Bank Sta=4229.9,4363.6
XS Rating Curve= 0 ,0
Exp/Cntr=0.3,0.1

Type RM Length L Ch R = 1 ,36353   ,342,342,342
BEGIN DESCRIPTION:
WOODSONS GULLY 71.0
END DESCRIPTION:
XS GIS Cut Line= 3
      3872102.94     10043324.84      3871611.21     10042796.86
      3871228.54     10041955.83
#Sta/Elev= 30
  4278.5   93.81  4362.7   91.43  4406.9   91.53  4454.6   91.09  4482.9   92.42
  4489.8   91.55  4582.1   91.86  4588.9   91.03  4617.3   91.26  4624.6   92.54
  4652.6    93.3  4723.3   91.76  4744.8   93.03  4786.7   91.61  4857.6   93.18
 4889.16  92.291    4971   90.75  4994.1   88.97  5021.5   90.74  5067.6   90.63
  5083.3   92.36  5188.4   94.15  5226.1   92.79  5354.5    95.7  5467.8   93.68
  5709.5   96.69  5769.3    96.5  5775.4   97.48  5890.1    97.6    5924   99.14
#Mann= 6 ,-1 , 0
  4278.5     .05       0  4406.9     .12       0  4786.7      .1       0
 4889.16     .03       0  5083.3      .1       0  5354.5     .12       0
Bank Sta=4889.16,5083.3
XS Rating Curve= 0 ,0
Exp/Cntr=0.3,0.1

Type RM Length L Ch R = 1 ,36011   ,511,511,511
BEGIN DESCRIPTION:
WOODSONS GULLY 70.0
END DESCRIPTION:
XS GIS Cut Line= 3
       3872296.1     10043282.54      3871874.95     10042674.72
      3871496.58     10042435.72
#Sta/Elev= 30
  4348.3   94.65  4362.3   93.34  4398.8   93.87  4447.6   90.72    4549   93.06
  4683.8   93.52  4721.9   94.47  4736.8   93.15  4778.7   94.18 4792.38  93.292
  4865.2   90.65  4987.4   90.89  5003.7   88.93  5013.1   88.93  5017.2   90.66
  5031.4   90.52  5038.1   92.36    5053   93.24  5059.1   92.37  5124.2   93.83
  5160.7   93.19    5176   94.36  5181.9   93.52  5248.9    94.4  5320.9   92.13
  5327.7   93.22  5406.6   93.04  5427.8   94.53  5500.7   95.96  5535.3   95.17
#Mann= 4 ,-1 , 0
  4348.3     .05       0  4683.8     .12       0 4792.38     .03       0
    5053      .1       0
Bank Sta=4792.38,5053
XS Rating Curve= 0 ,0
Exp/Cntr=0.3,0.1

Type RM Length L Ch R = 1 ,35500   ,500,500,500
BEGIN DESCRIPTION:
WOODSONS GULLY 69.0
END DESCRIPTION:
XS GIS Cut Line= 3
      3872373.65     10042521.86      3872239.02     10042457.09
      3872001.77     10042280.27
#Sta/Elev= 30
  4850.6   94.09  4868.8   92.43    4894   92.16  4901.4   91.77  4923.6   92.73
  4931.2   91.88  4936.7   92.69 4940.92  92.333    4968   90.08    4982    90.3
    4985   89.75  4985.5   89.25  4994.9   89.25  4995.4   89.75  5004.7   90.74
  5013.1   90.28  5040.1   90.65  5063.1   90.24  5076.3   90.77  5119.4   90.03
    5134   92.45  5140.2    92.5  5148.6   93.33  5184.9   94.03  5193.7   93.69
    5226   93.86  5254.9   93.19  5275.8    93.3  5284.1   92.81  5295.9   94.02
#Mann= 6 ,-1 , 0
  4850.6     .05       0    4894      .1       0 4940.92     .03       0
    5134      .1       0  5184.9     .05       0  5193.7     .12       0
Bank Sta=4940.92,5134
XS Rating Curve= 0 ,0
Exp/Cntr=0.3,0.1

Type RM Length L Ch R = 1 ,35000   ,395,395,395
BEGIN DESCRIPTION:
WOODSONS GULLY 68.0
END DESCRIPTION:
XS GIS Cut Line= 3
      3872670.14      10042350.3      3872552.86     10042142.74
      3872464.06     10042015.82
#Sta/Elev= 30
  4761.6   94.15  4771.4   93.66  4783.7   94.02  4814.7   93.97  4820.5    93.6
  4829.6   93.99  4853.4   93.78  4864.1   93.99  4879.7   93.08  4887.1   93.35
  4901.3   92.57    4933   92.38 4942.31  91.668  4976.4    89.6  4990.4   90.38
  4998.1    89.6  5012.8   90.14  5039.8   89.47  5048.5   89.77  5049.9   88.95
  5059.4   88.95  5059.9   89.45  5063.1   90.03  5099.1   89.96  5105.2   90.56
  5111.9   91.85  5120.1   92.21  5126.2   92.02  5135.2   92.52  5154.9   93.18
#Mann= 5 ,-1 , 0
  4761.6     .05       0  4853.4     .12       0 4942.31     .03       0
  5111.9      .1       0  5135.2     .05       0
Bank Sta=4942.31,5111.9
XS Rating Curve= 0 ,0
Exp/Cntr=0.3,0.1

Type RM Length L Ch R = 1 ,34605   ,682,682,682
BEGIN DESCRIPTION:
WOODSONS GULLY 67.0
END DESCRIPTION:
XS GIS Cut Line= 3
      3872868.12     10042241.54      3872891.55     10042018.12
      3872912.39     10041856.31
#Sta/Elev= 30
    4764   93.93  4774.5    93.4  4784.6   93.26  4794.6   93.44  4804.5   93.08
  4809.5   93.39  4834.9   92.52    4865   91.94  4875.1   91.41  4895.2   91.09
  4902.7   90.22  4907.8   90.51  4915.3   90.14  4935.4   89.77  4945.5   90.17
  4965.6   90.08  4988.7   90.41  4994.8   89.62  4999.8   89.88  5001.1      89
  5010.6      89  5011.1    89.5  5015.9   89.71  5056.3   89.96 5083.25  93.133
  5086.5   93.62  5092.7   92.82  5096.6   92.32  5106.7   92.92  5151.8   93.99
#Mann= 4 ,-1 , 0
    4764     .05       0  4809.5     .03       0 5083.25      .1       0
  5092.7     .12       0
Bank Sta=4809.5,5083.25
XS Rating Curve= 0 ,0
Exp/Cntr=0.3,0.1

Type RM Length L Ch R = 1 ,33923   ,375,375,375
BEGIN DESCRIPTION:
WOODSONS GULLY 66.0
END DESCRIPTION:
XS GIS Cut Line= 3
      3873244.25      10042571.4      3873266.47     10042374.19
      3873244.33     10042134.16
#Sta/Elev= 30
  4814.3   94.39    4817   94.39  4824.7    93.3  4844.8   92.48  4864.9   92.16
  4885.1   92.82  4915.3   90.28  4935.4   89.48  4945.4   90.28  4955.5   89.71
  4975.5   89.63  4980.5   89.22    4981   88.72  4990.5   88.72    4991   89.22
  4995.8   89.76  5011.8   90.25    5046   90.18  5051.6   90.45  5056.6   90.01
  5066.1   89.93  5096.2   90.79  5136.4   90.22  5146.4   90.79  5161.3      91
  5186.4   92.46  5196.6   92.62  5206.7   92.21  5226.8   92.52  5253.8   93.74
#Mann= 3 , 0 , 0
  4814.3     .05       0  4885.1     .03       0  5186.4      .1       0
Bank Sta=4885.1,5186.4
XS Rating Curve= 0 ,0
Exp/Cntr=0.3,0.1

Type RM Length L Ch R = 1 ,33548   ,548,548,548
BEGIN DESCRIPTION:
WOODSONS GULLY 65.0
END DESCRIPTION:
XS GIS Cut Line= 3
      3873770.23     10042330.61       3873491.6     10042229.05
      3873285.83     10042101.43
#Sta/Elev= 30
  4710.5   93.21  4734.3   91.66    4745   92.04  4756.9   90.54  4776.9   89.86
  4782.2   90.44  4819.5   90.21  4873.9   90.93  4893.8   91.91  4899.1   91.43
  4904.6   90.05  4915.3   90.98  4924.4   90.21  4929.7   90.53  4947.2   89.99
  5036.3   89.97  5040.5   89.48    5041   88.98  5050.5   88.98  5051.7   89.62
  5058.5   89.97  5082.1   90.36  5088.3   90.43  5094.2   89.61  5117.4   89.89
  5124.9   90.93  5140.3   91.81    5178   92.34  5235.1    92.7  5249.2    93.9
#Mann= 5 ,-1 , 0
  4710.5     .05       0  4893.8     .03       0  5140.3      .1       0
    5178     .12       0  5235.1      .1       0
Bank Sta=4893.8,5140.3
XS Rating Curve= 0 ,0
Exp/Cntr=0.3,0.1

Type RM Length L Ch R = 1 ,33000   ,474,474,474
BEGIN DESCRIPTION:
WOODSONS GULLY 64.0
END DESCRIPTION:
XS GIS Cut Line= 3
      3873492.65     10041683.08      3873368.09     10041806.71
      3873192.49     10041979.99
#Sta/Elev= 30
  4824.5    93.3  4840.6   92.74  4854.8   92.97  4861.8   92.15  4890.1   91.81
  4904.2   92.48  4925.5   91.84  4946.7   92.45  4968.5   92.34  4989.1   89.86
  4996.2   90.31  4999.5   89.59  5024.5   90.15  5038.6   89.92  5045.6   90.48
  5059.8   90.12  5062.2   89.09  5071.7   89.09  5072.2   89.59  5073.9   89.89
  5123.5   90.16  5137.6   91.06  5144.7   90.29  5158.8   90.45  5165.9   91.76
  5172.9   91.16  5187.1   92.43  5194.2   92.27  5208.3   93.22  5246.7   94.26
#Mann= 3 , 0 , 0
  4824.5     .12       0  4968.5     .03       0  5187.1     .12       0
Bank Sta=4968.5,5187.1
XS Rating Curve= 0 ,0
Exp/Cntr=0.3,0.1

Type RM Length L Ch R = 1 ,32526   ,477,477,477
BEGIN DESCRIPTION:
WOODSONS GULLY 63.0
END DESCRIPTION:
XS GIS Cut Line= 3
      3873396.47     10041443.53      3873161.67      10041450.9
      3872983.88     10041596.17
#Sta/Elev= 30
  4861.7   94.17  4938.6    91.6    4944   91.97  4950.4   91.26  4955.6    88.7
  4965.1    88.7  4965.6    89.2  4970.4   89.55  4980.4   89.81  5000.4   89.46
  5030.4    90.1  5070.4   90.23  5080.4   89.65  5106.4   89.67  5127.4    90.2
  5135.1   89.67  5141.6   90.21  5149.5   89.59  5163.8   89.96  5170.3   89.63
  5184.6   90.95    5199   90.47  5213.4   90.56  5219.8   90.12  5234.2   90.99
 5240.12  92.271  5242.1    92.7  5262.9   92.47  5291.6   93.88  5326.2   93.89
#Mann= 4 ,-1 , 0
  4861.7     .12       0  4938.6      .1       0    4944     .03       0
 5240.12     .12       0
Bank Sta=4944,5240.12
XS Rating Curve= 0 ,0
Exp/Cntr=0.3,0.1

Type RM Length L Ch R = 1 ,32049   ,490,490,490
BEGIN DESCRIPTION:
WOODSONS GULLY 62.0
END DESCRIPTION:
XS GIS Cut Line= 3
      3873487.58     10041103.69      3873272.78     10041144.05
      3873096.78     10041216.52
#Sta/Elev= 30
  4783.7   94.08  4786.1   94.08  4792.6   92.53  4797.6   93.13  4803.8   91.85
  4834.3   90.91  4855.2   89.68  4885.2      90  4895.4   89.63  4907.8   90.17
  4936.1    89.6  4955.2   90.01  4966.6   89.79  4971.5   89.43    4972   88.93
  4981.5   88.93    4982   89.43  4986.9   89.76  5004.9   89.55  5028.8   90.31
  5034.2   89.98    5040    90.6  5050.9   89.98  5087.5   89.73  5111.5   92.08
  5126.6   91.95  5164.8   92.74  5170.2   92.44  5180.6   93.45  5192.6   93.89
#Mann= 3 , 0 , 0
  4783.7     .12       0  4803.8     .03       0  5111.5     .12       0
Bank Sta=4803.8,5111.5
XS Rating Curve= 0 ,0
Exp/Cntr=0.3,0.1

Type RM Length L Ch R = 1 ,31559   ,559,559,559
BEGIN DESCRIPTION:
WOODSONS GULLY 61.0
END DESCRIPTION:
XS GIS Cut Line= 3
      3873017.32     10040807.12      3872975.65     10040972.07
      3873017.85     10041211.04
#Sta/Elev= 30
    4825   93.04  4838.7   93.14    4860   92.39  4870.3   91.48  4884.9   91.48
    4891   91.77  4901.3   89.97  4911.6   89.77  4920.8   90.29    4967   89.93
  5009.1   89.27  5009.6   88.77  5019.2   88.77  5019.7   89.27  5038.2   89.54
  5044.9   90.59    5055   89.79  5065.2   89.59  5075.4   90.07  5092.3   89.89
  5097.4   90.11    5116   91.99  5126.1   92.56  5146.4   93.34  5151.5   92.62
  5156.6   92.94  5187.1   92.96  5210.8   93.67  5227.7    93.8  5237.8   93.37
#Mann= 3 , 0 , 0
    4825      .1       0    4860     .03       0  5126.1     .12       0
Bank Sta=4860,5126.1
XS Rating Curve= 0 ,0
Exp/Cntr=0.3,0.1

Type RM Length L Ch R = 1 ,31000   ,500,500,500
BEGIN DESCRIPTION:
WOODSONS GULLY 60.0
END DESCRIPTION:
XS GIS Cut Line= 3
      3872506.14     10040977.52      3872610.06     10041155.04
      3872821.25     10041442.38
#Sta/Elev= 30
  4794.3    93.8  4799.3    93.8  4821.6   91.37  4843.1   91.61  4856.4   89.58
    4886   89.14  4891.8   89.77  4937.5    90.1  4950.5   89.25  4960.4    89.3
  4961.4   88.54    4971   88.54  4972.2   89.11    5003   89.17  5009.2    89.8
  5032.3   89.48  5044.7   90.62  5053.1   92.24  5059.4   91.67  5082.2   92.53
  5103.3   91.46  5203.6   90.94  5218.2    90.2  5224.4   90.77  5230.9   90.34
  5268.1      91  5303.9   90.18  5317.7   91.53    5331    91.4  5356.6   93.53
#Mann= 4 ,-1 , 0
  4794.3      .1       0  4843.1     .03       0  5053.1      .1       0
  5082.2     .12       0
Bank Sta=4843.1,5053.1
XS Rating Curve= 0 ,0
Exp/Cntr=0.3,0.1

Type RM Length L Ch R = 1 ,30500   ,707,707,707
BEGIN DESCRIPTION:
WOODSONS GULLY 59.0
END DESCRIPTION:
XS GIS Cut Line= 3
      3872323.86     10040881.15      3872194.67     10041116.86
      3872284.78      10041342.1
#Sta/Elev= 30
  4731.2   93.99  4742.5   93.96  4751.2   93.42  4778.7   90.94  4788.1   90.81
  4794.8   91.62  4810.9   90.09  4816.6   89.06  4854.5   89.61  4876.3   89.14
  4890.8   89.51  4903.8   89.15  4908.3    88.8  4908.8    88.3  4918.4    88.3
  4919.9   89.01  4941.7   89.07  4947.8   89.71  4957.8   89.92  4979.6   88.88
  5026.7   89.76  5104.8   88.92    5123   89.18  5134.4   89.88  5158.7   90.12
  5176.9   91.47  5207.1   91.75  5236.8   93.03    5240   93.67  5242.6   93.67
#Mann= 3 , 0 , 0
  4731.2      .1       0  4794.8     .03       0  5176.9      .1       0
Bank Sta=4794.8,5176.9
XS Rating Curve= 0 ,0
Exp/Cntr=0.3,0.1

Type RM Length L Ch R = 1 ,29793   ,305,305,305
BEGIN DESCRIPTION:
WOODSONS GULLY 58.0
END DESCRIPTION:
XS GIS Cut Line= 3
      3871743.12      10040649.4      3871619.42     10040829.09
      3871316.03     10041232.74
#Sta/Elev= 30
  4734.6   93.57  4738.9   93.82  4747.7   92.02  4753.8   92.72  4760.9    92.2
  4804.5   92.51  4810.6   93.27  4833.7   91.93  4861.3   88.74  4968.8   89.12
  4986.3   88.61  4986.8   88.11  4996.6   88.11    4998    88.9  5155.4   89.42
  5183.4   91.63  5197.9   92.31  5212.5      92  5223.6   92.62  5255.5   92.86
  5262.5   93.49  5297.9   92.43  5312.5   93.71  5327.1   93.46  5391.6   95.23
  5405.6   95.18    5427   96.21  5447.9   96.36  5453.5   97.62  5457.7   97.62
#Mann= 4 ,-1 , 0
  4734.6      .1       0  4833.7     .03       0  5183.4      .1       0
  5223.6     .12       0
Bank Sta=4833.7,5183.4
XS Rating Curve= 0 ,0
Exp/Cntr=0.3,0.1

Type RM Length L Ch R = 1 ,29488   ,488,488,488
BEGIN DESCRIPTION:
WOODSONS GULLY 57.0
END DESCRIPTION:
XS GIS Cut Line= 3
      3871547.83     10040497.02      3871308.22     10040830.39
      3871064.72     10041099.94
#Sta/Elev= 30
  4593.8    93.1  4697.3    91.2    4719   89.98  4740.4   89.72  4754.6   88.95
  4769.4   89.41  4775.5   91.25  4790.2   90.18  4796.4   90.95  4832.8   90.45
  4840.6      91  4846.7   90.27  4876.2   91.07  4905.6   90.55    4919   91.24
  4932.7   91.02  4941.2   90.12  4947.4   91.05  4955.9   88.79  4991.6   88.96
  4992.8   88.26  5097.4   91.19  5132.5   91.52  5167.6    93.8  5237.9    95.3
  5288.2   96.65  5309.6   98.12  5316.3   97.43    5338    97.5  5367.6    98.9
#Mann= 6 ,-1 , 0
  4593.8      .1       0  4740.4     .12       0  4947.4     .03       0
  5097.4     .12       0  5237.9     .05       0  5288.2     .12       0
Bank Sta=4947.4,5097.4
XS Rating Curve= 0 ,0
Exp/Cntr=0.3,0.1

Type RM Length L Ch R = 1 ,29000   ,500,500,500
BEGIN DESCRIPTION:
WOODSONS GULLY 56.0
END DESCRIPTION:
XS GIS Cut Line= 3
      3871540.61     10040435.87      3871029.17     10040487.15
      3870651.77     10040642.44
#Sta/Elev= 30
    4486   92.41  4498.8   91.12  4518.9   91.49  4569.2   89.39  4619.4   88.71
  4760.1   89.19    4825   88.48  4825.5   87.98  4835.4   87.98  4850.6   89.47
  4860.6   89.11  4890.2  91.755  4892.4   92.32    4931   91.45  4961.1   88.53
  4971.2   89.04  4987.7   88.49  4992.7   89.23  5003.4   88.69  5049.9   89.81
  5066.3   89.42  5073.9   90.22  5079.3   89.88  5140.5   92.35  5180.5   94.16
  5217.7   94.72  5228.4   94.15  5271.8   96.25  5368.8   97.77  5408.1   98.84
#Mann= 5 ,-1 , 0
    4486      .1       0  4518.9     .03       0  4890.2      .1       0
  5140.5     .05       0  5368.8     .12       0
Bank Sta=4518.9,4890.2
XS Rating Curve= 0 ,0
Exp/Cntr=0.3,0.1

Type RM Length L Ch R = 1 ,28500   ,500,500,500
BEGIN DESCRIPTION:
WOODSONS GULLY 55.0
END DESCRIPTION:
XS GIS Cut Line= 3
      3871542.28      10040433.6      3870938.55     10040014.39
      3870611.67      10039938.4
#Sta/Elev= 30
    4265   92.41  4270.7   92.41  4277.3   91.38  4292.2    91.9  4319.2   90.96
  4334.1   91.61  4363.8   88.83  4471.2   88.06  4536.7   89.17  4542.8   88.19
  4572.5   88.33    4582   87.46  4591.9   87.46  4593.4   88.69  4644.1   88.04
  4757.5   88.37  4793.9   90.43  4816.9   90.14  4852.7    91.5  4873.7   92.43
  4924.3    92.4  4945.3   91.41  4960.1   89.29    4975    88.4    5052    89.7
  5093.1   91.59  5121.9   91.83  5137.8   93.33  5308.7   96.92  5335.6   96.68
#Mann= 4 ,-1 , 0
    4265      .1       0  4334.1     .03       0  4852.7      .1       0
  5137.8     .12       0
Bank Sta=4334.1,4852.7
XS Rating Curve= 0 ,0
Exp/Cntr=0.3,0.1

Type RM Length L Ch R = 1 ,28000   ,500,500,500
BEGIN DESCRIPTION:
WOODSONS GULLY 54.0
END DESCRIPTION:
XS GIS Cut Line= 3
      3871548.42     10040394.27      3871357.23     10039805.43
      3871302.81     10039458.88
#Sta/Elev= 30
  4380.9   91.86  4468.7   90.59  4500.6   88.15    4542    87.9  4559.3   89.24
  4564.6   88.21    4584   89.16  4605.1   88.05  4623.2   89.62  4636.6   88.41
  4678.7   88.08  4687.1   88.79  4705.2   87.31  4731.2   88.53  4804.8   88.11
  4820.2   88.56 4842.17  90.731  4916.1   93.16  4953.3   91.64    4980   88.76
  5034.8   88.48  5075.3   90.84  5115.8   91.01  5206.9   94.45  5221.8   94.19
  5318.2   97.16  5328.3   96.11  5338.8    96.2  5343.6    96.4  5350.8   96.94
#Mann= 5 ,-1 , 0
  4380.9      .1       0  4468.7     .03       0 4842.17      .1       0
  5338.8     .12       0  5343.6      .1       0
Bank Sta=4468.7,4842.17
XS Rating Curve= 0 ,0
Exp/Cntr=0.3,0.1

Type RM Length L Ch R = 1 ,27500   ,500,500,500
BEGIN DESCRIPTION:
WOODSONS GULLY 53.0
END DESCRIPTION:
XS GIS Cut Line= 3
      3872149.72     10040130.76      3871855.91     10039803.77
      3871571.65     10039520.08
#Sta/Elev= 30
  4560.4   93.35  4575.4   90.77  4632.2   89.37  4667.5   89.38  4674.8    90.2
    4781   89.31  4788.5   90.11  4816.1   88.94  4872.9   91.28  4880.4   90.67
  4901.3   91.49  4915.5   89.15  4929.7   88.16  4943.9   87.86  4950.7   88.73
  4958.1    87.9  5016.8   86.88    5043    88.2  5085.4      88  5127.8   89.75
  5177.3   90.21  5184.4   89.27    5248   91.53  5269.2   92.18  5304.6    95.1
  5325.8   94.18  5361.2   95.73  5371.8   95.22  5382.4   95.09  5401.6   96.92
#Mann= 4 ,-1 , 0
  4560.4      .1       0  4901.3     .03       0    5248      .1       0
  5371.8     .12       0
Bank Sta=4901.3,5248
XS Rating Curve= 0 ,0
Exp/Cntr=0.3,0.1

Type RM Length L Ch R = 1 ,27000   ,564,564,564
BEGIN DESCRIPTION:
WOODSONS GULLY 52.0
END DESCRIPTION:
XS GIS Cut Line= 3
      3872367.26     10039245.09      3872098.24     10039434.12
      3871696.21      10039422.2
#Sta/Elev= 30
  4671.2   92.35  4710.5   90.68  4725.3   89.83    4761   89.51  4775.8    88.7
  4804.9   88.65  4811.5   88.05  4817.7   88.47  4847.3   88.06  4853.8    88.6
  4862.1    87.9  4890.5   88.34  4927.1   87.41  4928.5   86.83  4938.6   86.83
  4939.6   87.57  4954.4   87.83  5010.4   87.47  5030.4   88.09  5060.4   87.66
  5070.4   88.07  5090.4   90.57  5110.4   90.62  5150.5   92.98  5260.5   91.99
  5273.6    92.9  5320.5    93.6  5360.5   95.07  5380.6   95.15  5402.2    96.2
#Mann= 3 , 0 , 0
  4671.2      .1       0  4710.5     .03       0  5090.4      .1       0
Bank Sta=4710.5,5090.4
XS Rating Curve= 0 ,0
Exp/Cntr=0.3,0.1

Type RM Length L Ch R = 1 ,26436   ,436,436,436
BEGIN DESCRIPTION:
WOODSONS GULLY 51.0
END DESCRIPTION:
XS GIS Cut Line= 3
      3872198.31     10038971.16      3871919.66     10038984.18
      3871685.51     10038946.02
#Sta/Elev= 30
  4719.6   93.61  4730.1   93.31  4740.1   91.95  4750.1   91.45  4770.1   91.99
    4820   91.53  4830.2   91.95  4850.2   91.28  4870.2   91.86  4890.2      90
  4900.3   90.46  4920.3   89.18  4930.3   89.21  4960.3   87.93  4980.3   87.96
  4984.8   87.56  4985.3   87.06  4995.4   87.06    4997   87.81  5052.5   88.52
  5071.3   90.28  5081.4   90.26 5105.86    91.8    5109   92.14    5114   91.72
    5122   92.07  5142.2   93.58  5182.8   94.64  5213.2   96.12  5235.8   96.48
#Mann= 3 , 0 , 0
  4719.6      .1       0  4870.2     .03       0 5105.86     .12       0
Bank Sta=4870.2,5105.86
XS Rating Curve= 0 ,0
Exp/Cntr=0.3,0.1

Type RM Length L Ch R = 1 ,26000   ,500,500,500
BEGIN DESCRIPTION:
WOODSONS GULLY 50.0
END DESCRIPTION:
XS GIS Cut Line= 3
      3872213.07     10038966.78      3872251.15     10038786.86
      3872245.87      10038408.6
#Sta/Elev= 30
  4816.1   94.14  4832.2   91.75  4860.5   90.34    4873   90.44  4893.5   89.49
 4928.82  89.058  4959.9   87.69  4989.7   87.21  4990.2   86.71  5000.3   86.71
  5000.8   87.21  5005.8   87.56  5035.8   87.94  5055.8   87.51  5105.8    89.3
  5115.8   88.92  5155.8   89.74  5195.8   90.78  5205.8   91.91  5225.8   91.55
  5235.8   92.21  5245.8   91.93  5255.8   92.75  5275.8   93.11  5305.8   93.25
  5315.8   92.83  5335.8   93.85  5345.8   93.53  5367.2   94.51  5378.3   94.91
#Mann= 4 ,-1 , 0
  4816.1      .1       0 4928.82     .03       0  5105.8      .1       0
  5367.2     .05       0
Bank Sta=4928.82,5105.8
XS Rating Curve= 0 ,0
Exp/Cntr=0.3,0.1

Type RM Length L Ch R = 1 ,25500   ,458,458,458
BEGIN DESCRIPTION:
WOODSONS GULLY 49.0
END DESCRIPTION:
XS GIS Cut Line= 3
      3872308.83     10039101.37      3872468.24      10039083.5
      3872623.11     10039017.13
#Sta/Elev= 30
  4839.6   92.09  4858.7    91.6  4868.8   91.18  4878.9   91.32  4885.5   90.94
  4890.6    90.9    4899   90.16    4909   90.22  4949.3    88.5  4959.4   87.67
  4969.4   88.19  4975.7   87.76  4980.7   87.88  4991.7    87.2  4992.2    86.7
  5002.3    86.7  5002.8    87.2  5032.2   87.22    5041    87.5  5046.4   87.23
  5064.5   88.89  5093.5   90.21  5108.4   90.11  5117.1   90.72  5130.1   91.14
  5140.7   91.87  5146.1   91.82  5151.9   92.84  5162.8   92.98  5168.5   92.53
#Mann= 3 , 0 , 0
  4839.6      .1       0    4909     .03       0  5093.5      .1       0
Bank Sta=4909,5093.5
XS Rating Curve= 0 ,0
Exp/Cntr=0.3,0.1

Type RM Length L Ch R = 1 ,25042   ,542,542,542
BEGIN DESCRIPTION:
WOODSONS GULLY 48.0
END DESCRIPTION:
XS GIS Cut Line= 3
       3872554.7      10039519.1       3872680.4     10039357.98
      3872742.72     10039095.53
#Sta/Elev= 30
  4794.5    90.9  4823.9    89.6  4830.2   88.55  4844.7   87.82  4859.1   87.61
  4880.8   87.96  4944.2   86.69  4966.8   87.29  4973.1   86.91  4998.9   86.81
  5004.6   86.57  5005.1   86.07  5015.4   86.07  5016.2   87.15  5036.8   87.12
  5047.1   87.96  5052.5   87.29  5067.6   87.22  5077.9    88.2  5088.2   88.57
  5094.7    89.5    5119   89.59    5142   90.43  5149.8   90.07  5160.1   90.19
  5201.2   91.34  5232.1   91.01  5252.6   91.21  5262.9   91.95  5268.6   91.74
#Mann= 3 , 0 , 0
  4794.5      .1       0  4823.9     .03       0  5094.7      .1       0
Bank Sta=4823.9,5094.7
XS Rating Curve= 0 ,0
Exp/Cntr=0.3,0.1

Type RM Length L Ch R = 1 ,24500   ,506,506,506
BEGIN DESCRIPTION:
WOODSONS GULLY 47.0
END DESCRIPTION:
XS GIS Cut Line= 3
      3873128.87     10039293.94       3873139.9     10039196.86
      3873170.31     10038984.53
#Sta/Elev= 30
  4902.3   89.63  4925.3   89.89    4934   90.17    4939   89.57  4945.4   88.63
  4955.5   87.57  4959.9   86.79  4960.4   86.29  4970.7   86.29  4971.2   86.79
  4985.7   87.06  5005.9   87.03  5015.9   87.12  5020.9      87  5056.4    87.3
  5076.6   87.14  5091.5   87.47  5096.8   88.05  5106.9    88.5    5117   89.34
  5127.1   89.52  5137.2   90.43  5147.3   90.09  5157.1   90.34  5162.2   90.32
  5167.5   90.78  5187.7      92  5197.8   92.14  5207.9   92.93  5214.5   93.05
#Mann= 3 , 0 , 0
  4902.3      .1       0    4934     .03       0  5137.2      .1       0
Bank Sta=4934,5137.2
XS Rating Curve= 0 ,0
Exp/Cntr=0.3,0.1

Type RM Length L Ch R = 1 ,23994   ,494,494,494
BEGIN DESCRIPTION:
WOODSONS GULLY 46.0
END DESCRIPTION:
XS GIS Cut Line= 3
      3873485.64     10039518.01      3873546.59     10039298.19
      3873541.42       10039155.
#Sta/Elev= 30
  4768.8   90.04  4793.7   89.86  4798.9   89.69  4807.1    88.8  4838.3   88.29
    4859   88.12  4867.4   88.27  4872.6   87.97  4890.1   88.25  4900.5   88.09
  4912.1   87.02  4921.3   86.98    4926   86.38  4926.5   85.88  4936.8   85.88
  4937.3   86.38  4941.2   86.57  4952.4   86.48  4980.6   86.85  4985.8    87.1
  4992.8   86.55    5014   86.76  5034.1   86.62  5054.1   87.16  5064.1   87.97
  5074.1   87.98 5078.84  88.383  5094.1   89.49  5099.8   90.27  5140.2   90.97
#Mann= 3 , 0 , 0
  4768.8      .1       0  4900.5     .03       0 5078.84      .1       0
Bank Sta=4900.5,5078.84
XS Rating Curve= 0 ,0
Exp/Cntr=0.3,0.1

Type RM Length L Ch R = 1 ,23500   ,500,500,500
BEGIN DESCRIPTION:
WOODSONS GULLY 45.0
END DESCRIPTION:
XS GIS Cut Line= 3
      3873782.77     10039607.83      3873887.35     10039476.86
      3873964.15     10039323.18
#Sta/Elev= 30
  4832.4   90.81    4848   90.37  4854.4   89.71  4862.4   90.12  4876.8   90.07
 4879.93   89.38  4883.2   88.66  4897.6    86.8    4905   86.98  4955.3   86.45
    4956   86.27  4956.5   85.77  4966.8   85.77  4967.3   86.27    4969   86.43
  4982.5    86.6  4990.5   86.31  5006.5   86.56  5028.8    86.3  5040.1   86.69
  5051.2   86.65  5062.5   88.38  5079.3   89.45  5095.9   89.53  5098.7   89.26
  5101.6   88.99    5124   90.05  5146.4   89.71    5152   90.03  5171.8   90.31
#Mann= 4 ,-1 , 0
  4832.4      .1       0 4879.93     .03       0  5079.3      .1       0
  5098.7     .12       0
Bank Sta=4879.93,5079.3
XS Rating Curve= 0 ,0
Exp/Cntr=0.3,0.1

Type RM Length L Ch R = 1 ,23000   ,500,500,500
BEGIN DESCRIPTION:
WOODSONS GULLY 44.0
END DESCRIPTION:
XS GIS Cut Line= 3
      3874444.67     10039705.74      3874188.24     10039418.16
      3874053.57     10039360.47
#Sta/Elev= 30
  4614.7   91.14    4651   89.99  4658.5    90.1  4665.2   89.55  4679.4   90.08
  4686.9   89.33  4707.8   89.31  4714.7    88.7  4750.4   90.18  4807.3   89.78
  4821.5   88.91  4828.2   89.26  4842.4   88.82  4849.1   88.04  4856.6   88.03
  4863.3   86.66  4870.8   87.39  4877.5   86.56  4920.2   86.24  4955.9   86.88
  5022.2   86.26  5023.5   86.13    5024   85.63  5034.4   85.63  5034.9   86.13
  5052.7   86.95  5065.7   88.64  5087.5   89.59    5139   90.65  5146.5   90.72
#Mann= 4 ,-1 , 0
  4614.7      .1       0  4807.3     .03       0  5087.5      .1       0
    5139     .12       0
Bank Sta=4807.3,5087.5
XS Rating Curve= 0 ,0
Exp/Cntr=0.3,0.1

Type RM Length L Ch R = 1 ,22500   ,613,613,613
BEGIN DESCRIPTION:
WOODSONS GULLY 43.0
END DESCRIPTION:
XS GIS Cut Line= 3
      3874602.86     10039463.38      3874540.66     10039236.86
      3874549.68     10038986.03
#Sta/Elev= 30
  4765.1   90.65  4788.2    90.6  4798.2   90.27  4803.3   90.49    4809   89.74
  4819.3   89.75  4829.7   89.23    4843   89.43  4871.2   88.52  4877.4   89.32
  4882.6   88.91  4896.7  88.478  4902.3   88.22  4911.8   87.28    4917   88.03
    4923   86.61  4933.4   86.13  4964.5   86.61  4985.3   86.13  5035.8   86.37
  5055.2      86  5055.7    85.5  5066.1    85.5  5066.6      86  5145.9   87.17
  5175.9   88.55  5195.9   88.52  5225.9    88.7  5235.9   89.06    5251   90.25
#Mann= 4 ,-1 , 0
  4765.1      .1       0  4896.7     .03       0  5175.9      .1       0
  5195.9     .12       0
Bank Sta=4896.7,5175.9
XS Rating Curve= 0 ,0
Exp/Cntr=0.3,0.1

Type RM Length L Ch R = 1 ,21887   ,387,387,387
BEGIN DESCRIPTION:
WOODSONS GULLY 42.0
END DESCRIPTION:
XS GIS Cut Line= 3
      3875189.64     10039194.61      3875028.24     10039184.85
      3874888.01      10039116.5
#Sta/Elev= 30
  4838.3   90.82  4841.7   90.82  4850.1   90.37  4860.1   90.04  4890.2   89.83
  4898.8   89.61  4930.3   88.63  4950.3    86.4  4977.5   86.08  4990.4   86.53
  4997.7   86.02    5003   86.02  5011.6    86.3  5018.6   85.91  5033.8   85.93
  5041.1   86.51  5046.7   86.45  5057.8   85.87  5058.3   85.37    5069   85.37
  5069.5   85.87  5091.7   86.52  5100.5   86.49  5108.7   86.31  5114.3   86.91
  5122.8   88.47  5131.3   89.26  5136.8   89.97    5145   90.62    5156   90.58
#Mann= 4 ,-1 , 0
  4838.3     .12       0  4898.8      .1       0  4930.3     .03       0
  5122.8     .12       0
Bank Sta=4930.3,5122.8
XS Rating Curve= 0 ,0
Exp/Cntr=0.3,0.1

Type RM Length L Ch R = 1 ,21500   ,504,504,504
BEGIN DESCRIPTION:
WOODSONS GULLY 41.0
END DESCRIPTION:
XS GIS Cut Line= 3
      3875233.06     10039142.58      3875184.21     10038922.84
       3875102.3     10038810.17
#Sta/Elev= 30
  4774.9   90.33  4778.7    90.5  4796.9      90  4822.2   89.92  4848.2   88.29
  4865.8   88.65    4876   88.34  4889.1   87.97  4909.3   86.05  4914.4    86.2
  4919.9   86.84  4930.1   86.28  4940.3    86.1  4950.6   86.13  4963.1   86.83
  4981.3   86.08  4998.3   85.96  4999.5   85.76    5000   85.26  5010.7   85.26
  5011.2   85.76  5013.8   85.91  5034.7   86.13  5040.9   86.64    5064   86.12
  5070.3   86.34  5091.1   86.17  5099.6   87.57 5107.25  88.197  5139.3   89.98
#Mann= 4 ,-1 , 0
  4774.9     .12       0    4876      .1       0  4889.1     .03       0
 5107.25      .1       0
Bank Sta=4889.1,5107.25
XS Rating Curve= 0 ,0
Exp/Cntr=0.3,0.1

Type RM Length L Ch R = 1 ,20996   ,396,396,396
BEGIN DESCRIPTION:
WOODSONS GULLY 40.0
END DESCRIPTION:
XS GIS Cut Line= 3
      3875597.27     10039152.84      3875575.57     10038850.76
      3875251.89     10038720.94
#Sta/Elev= 30
  4538.4   90.66  4550.2   89.59  4569.3   88.97  4580.3   89.23  4597.7   88.28
  4602.7   88.69  4626.5   87.35  4660.5   86.51  4670.5   87.32  4690.6   86.24
  4737.7   85.79  4742.7   86.65  4770.8   87.23  4854.4   87.23  4860.3   86.23
    4884   85.79    4962   86.17  4991.6   85.93  4995.1   85.23  5005.8   85.23
  5006.3   85.73    5022   86.38    5040   86.33  5045.4   85.74  5069.6   86.54
 5081.62  87.569  5099.2   88.78  5123.4   88.41    5162   89.67    5190   89.89
#Mann= 5 ,-1 , 0
  4538.4      .1       0  4569.3     .05       0  4626.5      .1       0
  4854.4     .03       0 5081.62      .1       0
Bank Sta=4854.4,5081.62
XS Rating Curve= 0 ,0
Exp/Cntr=0.3,0.1

Type RM Length L Ch R = 1 ,20600   ,508,508,508
BEGIN DESCRIPTION:
WOODSONS GULLY 39.0
END DESCRIPTION:
XS GIS Cut Line= 3
      3875243.82     10038374.38      3875184.77     10038548.74
      3875185.46     10038687.56
#Sta/Elev= 30
  4817.9   89.87  4820.3   89.42  4825.6   90.08  4835.5   89.76  4846.1   88.87
  4851.7   89.29    4857    88.9  4867.2   88.38  4877.7   88.23  4883.1   87.34
  4898.9   86.18  4914.6   86.09    4920   85.59  4930.5   85.78  4962.2   85.77
  4977.4   85.88  4993.9   85.64  4994.7   85.55  4995.2   85.05  5005.9   85.05
  5006.4   85.55  5024.3    85.8  5064.3   85.61  5074.3   86.11  5084.3   87.63
  5094.3      88  5104.3   88.86  5124.3   89.15  5134.3   89.58  5140.8   89.51
#Mann= 3 , 0 , 0
  4817.9      .1       0  4877.7     .03       0  5084.3      .1       0
Bank Sta=4877.7,5084.3
XS Rating Curve= 0 ,0
Exp/Cntr=0.3,0.1

Type RM Length L Ch R = 1 ,20092   ,592,592,592
BEGIN DESCRIPTION:
WOODSONS GULLY 38.0
END DESCRIPTION:
XS GIS Cut Line= 3
      3874745.89     10038382.05      3874716.02     10038607.77
      3874618.83     10038750.78
#Sta/Elev= 30
  4793.4   89.42    4812   88.42  4817.1   88.37  4822.7    89.3  4842.9   88.69
  4873.1   88.61 4875.32  88.276  4890.5   85.78  4903.4   85.86  4913.5   86.23
  4933.6   85.53  4953.8   86.06  4963.9   85.58  4978.2   85.37  4978.7   84.87
  4989.4   84.87  4989.9   85.37  5058.8   85.68  5064.9   86.17  5073.4   86.13
  5079.8   86.44  5085.8   86.08  5109.7   88.43  5117.7   88.39  5145.6   88.81
  5151.6   88.62  5166.6   89.11  5172.6   88.88  5191.2   90.44    5194   90.44
#Mann= 4 ,-1 , 0
  4793.4      .1       0 4875.32     .03       0  5109.7      .1       0
  5117.7     .12       0
Bank Sta=4875.32,5109.7
XS Rating Curve= 0 ,0
Exp/Cntr=0.3,0.1

Type RM Length L Ch R = 1 ,19500   ,599,599,599
BEGIN DESCRIPTION:
WOODSONS GULLY 37.0
END DESCRIPTION:
XS GIS Cut Line= 3
      3874729.82     10038286.67      3874558.24     10038258.36
      3874031.81     10038018.72
#Sta/Elev= 30
  4826.1   90.11  4848.4   88.16    4899   86.98  4909.2   85.34  4948.6   86.24
  4953.7   85.34  4959.8   86.72    4970   87.25  4997.7   85.35  5022.4   86.31
  5028.4   85.26  5028.9   84.76  5080.4    86.2  5103.4   85.66  5110.3   86.29
    5121   85.84  5132.3   86.31  5149.5   85.36    5155    86.4  5165.2   85.94
  5195.7   85.94  5201.1   86.44  5209.2   85.97  5224.2   86.43  5275.8   86.29
  5293.4   86.94  5362.5    86.7  5442.7   91.13  5549.8   94.97  5578.4   96.78
#Mann= 3 , 0 , 0
  4826.1      .1       0  5022.4     .03       0  5080.4     .12       0
Bank Sta=5022.4,5080.4
XS Rating Curve= 0 ,0
Exp/Cntr=0.3,0.1

Type RM Length L Ch R = 1 ,18901   ,514,514,514
BEGIN DESCRIPTION:
WOODSONS GULLY 36.0
END DESCRIPTION:
XS GIS Cut Line= 3
      3874589.15     10037767.62      3874544.62     10037778.48
      3874233.22     10037771.97
#Sta/Elev= 30
  4949.3   89.99  4952.6   89.99  4960.9   89.32  4971.2   88.73  4980.7   87.28
  4985.8   86.73  4990.9   85.58  4995.1   85.58  4996.5   84.35  5007.3   84.35
  5007.8   84.85  5021.9   85.71  5041.9   84.85  5071.9   85.38  5091.9   85.11
  5108.7   85.25  5113.7   85.13  5121.9   85.64  5131.9   85.33  5141.9   85.24
  5151.9    85.5  5191.9   88.76  5193.3   88.82  5201.9   89.19  5211.9   89.95
    5242   93.11    5252   93.71    5282   94.26    5292   94.82  5306.6   95.13
#Mann= 4 ,-1 , 0
  4949.3      .1       0  4971.2     .03       0  5191.9      .1       0
  5193.3     .12       0
Bank Sta=4971.2,5191.9
XS Rating Curve= 0 ,0
Exp/Cntr=0.3,0.1

Type RM Length L Ch R = 1 ,18387   ,335,335,335
BEGIN DESCRIPTION:
WOODSONS GULLY 35.0
END DESCRIPTION:
XS GIS Cut Line= 3
      3874847.36      10037494.2      3874492.97     10037376.01
      3874199.87     10037536.84
#Sta/Elev= 30
  4844.7   89.21  4886.3   88.61  4902.1   87.57  4907.4   88.13  4928.4    86.7
  4933.7   87.15    4960   85.42  5044.5    85.3    5049   84.78  5049.5   84.28
  5060.3   84.28  5060.8   84.78  5065.6   85.09  5107.7   85.34  5128.8    87.5
  5149.7   88.08  5202.6   88.68  5218.2   89.38  5224.1   88.61  5246.9   88.88
  5256.3   88.18  5299.9   87.95  5327.4   86.72  5395.2   86.29    5425   88.74
  5430.7   88.16  5440.8   88.42  5497.9   93.47  5506.5   93.22  5552.6    95.2
#Mann= 3 , 0 , 0
  4844.7     .12       0  4907.4     .03       0  5149.7     .12       0
Bank Sta=4907.4,5149.7
XS Rating Curve= 0 ,0
Exp/Cntr=0.3,0.1

Type RM Length L Ch R = 1 ,18052   ,552,552,552
BEGIN DESCRIPTION:
WOODSONS GULLY 34.0
END DESCRIPTION:
XS GIS Cut Line= 3
      3874845.08     10037095.78      3874440.18     10037288.86
      3874164.76     10037519.31
#Sta/Elev= 30
    4793   89.11  4900.7   87.43  4913.6   86.03  4936.3   85.24  5027.1   85.23
  5038.8   84.28  5072.5   85.18 5105.13  87.509  5117.8   87.54    5125   88.43
  5155.5   87.99  5177.7   89.22  5191.5   88.62  5246.4   90.22    5252   89.31
  5287.1   89.16  5294.9   87.62  5301.4   88.12  5309.2   86.99  5330.1   88.68
  5401.1   86.39  5436.7   87.16  5479.3   89.21  5492.7   90.48  5500.5   90.29
  5529.1   93.11  5543.4   93.83    5550   93.24  5557.5   94.27  5600.7   96.54
#Mann= 4 ,-1 , 0
    4793      .1       0  4900.7     .03       0 5105.13      .1       0
    5125     .12       0
Bank Sta=4900.7,5105.13
XS Rating Curve= 0 ,0
Exp/Cntr=0.3,0.1

Type RM Length L Ch R = 1 ,17500   ,406,406,406
BEGIN DESCRIPTION:
WOODSONS GULLY 33.0
END DESCRIPTION:
XS GIS Cut Line= 3
      3875086.72     10037251.57      3874852.78     10036832.32
       3873998.4     10036416.04
#Sta/Elev= 30
  4519.9    89.3    4543   87.65  4577.7   87.34  4592.2   88.13  4608.1   87.11
  4795.7   87.12  4819.5   87.25  4851.5   86.06  4954.4   85.79  4960.1   84.75
  4984.4   83.99  4995.5   83.99  4999.9   85.42 5023.73  87.259    5050   88.33
  5102.8   88.34    5139   86.94    5228   86.97  5288.7   88.64  5417.1   87.22
    5452   87.81    5469    89.2  5550.5   87.96  5587.3    85.4  5653.1   85.55
  5706.3   86.72  5739.5   85.16  5795.7   85.56  5880.3   93.21  5950.4   96.17
#Mann= 5 ,-1 , 0
  4519.9      .1       0  4795.7     .12       0  4819.5     .03       0
 5023.73      .1       0  5653.1      .1       0
Bank Sta=4819.5,5023.73
XS Rating Curve= 0 ,0
Exp/Cntr=0.3,0.1

Type RM Length L Ch R = 1 ,17094   ,484,484,484
BEGIN DESCRIPTION:
WOODSONS GULLY 32.0
END DESCRIPTION:
XS GIS Cut Line= 3
      3875114.26      10037212.3       3875058.7     10036583.78
      3874082.13     10036340.02
#Sta/Elev= 30
  4338.2   89.18  4369.5   87.68  4419.7    87.8  4459.9   86.84  4471.3   87.59
  4629.8   86.59  4821.3    85.3  4871.5   86.96  4972.2   85.49  4985.1   83.53
  5021.6   84.22    5051  87.046  5062.8    87.8  5080.9   86.96  5122.2   87.91
    5155   87.02  5217.4   87.81  5320.5   86.15  5402.9      89  5485.4   87.72
  5498.7   86.04  5568.2   85.53  5665.4   85.06  5732.7   85.44  5763.7   86.62
  5823.6   85.27  5835.8    86.7  5897.7   88.69  5938.9   92.75  5975.7   94.39
#Mann= 7 ,-1 , 0
  4338.2      .1       0  4629.8     .12       0  4871.5     .07       0
    5051      .1       0    5155     .12       0  5568.2     .05       0
  5665.4      .1       0
Bank Sta=4871.5,5051
XS Rating Curve= 0 ,0
Exp/Cntr=0.3,0.1

Type RM Length L Ch R = 1 ,16610   ,610,610,610
BEGIN DESCRIPTION:
WOODSONS GULLY 31.0
END DESCRIPTION:
XS GIS Cut Line= 4
       3875263.9     10036931.81       3875256.3     10036785.28
      3875417.32     10036651.94      3875492.34     10036489.41
#Sta/Elev= 30
  4627.6   87.53  4645.6   87.23  4658.4   87.61  4688.4   86.58  4708.4   87.12
  4718.5   86.25  4728.5   86.16  4792.3   86.63    4821   85.85  4852.3   85.79
  4878.3   85.39  4913.4   85.84  4942.1      85  4948.6    83.9  4970.8   83.95
  4977.3   83.44  4986.6      84  4998.7    83.6  5000.8   82.77  5011.9   82.77
  5012.4   83.27  5021.7   84.42  5028.4   83.52  5044.6   83.84  5050.4   84.49
  5083.5      85    5096   85.87  5105.5   85.87  5127.5   87.59  5162.4   87.79
#Mann= 4 ,-1 , 0
  4627.6     .12       0  4852.3      .1       0  4913.4     .03       0
    5096      .1       0
Bank Sta=4913.4,5096
XS Rating Curve= 0 ,0
Exp/Cntr=0.3,0.1

Type RM Length L Ch R = 1 ,16000   ,500,500,500
BEGIN DESCRIPTION:
WOODSONS GULLY 30.0
END DESCRIPTION:
XS GIS Cut Line= 3
      3875838.66     10036501.08      3875698.24     10036511.39
      3875556.04     10036486.84
#Sta/Elev= 30
  4859.2   86.83  4862.1   86.83    4870   86.43    4889   86.04  4900.1   86.15
  4910.1   85.76 4915.23  85.257  4926.3    84.3  4931.3   84.47  4940.2   83.73
  4950.3   83.47  4960.3    83.8  4970.3   83.45  4980.3   82.95  4990.4      83
  4991.6   82.57  4992.1   82.07  5003.2   82.07  5003.7   82.57  5010.5   83.13
  5020.7   83.03  5028.5   82.81    5041   83.98  5051.1    84.4  5061.3   85.17
  5081.6   85.34  5088.3   85.81    5112   87.06  5122.2    87.3  5144.3   87.49
#Mann= 4 ,-1 , 0
  4859.2     .12       0    4889      .1       0 4915.23     .03       0
  5061.3      .1       0
Bank Sta=4915.23,5061.3
XS Rating Curve= 0 ,0
Exp/Cntr=0.3,0.1

Type RM Length L Ch R = 1 ,15500   ,526,526,526
BEGIN DESCRIPTION:
WOODSONS GULLY 29.0
END DESCRIPTION:
XS GIS Cut Line= 3
       3875954.2      10036218.7      3875728.24     10036104.24
      3875607.28     10036084.84
#Sta/Elev= 30
  4746.7   86.78    4765   86.61  4772.6    86.1  4787.4   85.92  4817.2   84.12
  4822.8   84.94  4854.7   85.63  4861.7   85.12  4867.3   85.43  4877.1    84.8
  4899.5   84.41  4906.3   83.36  4911.9   83.34    4922   82.36  4933.3   83.71
  4934.2   83.81  4956.4   82.53  4966.8    82.4  4967.6   81.74  4978.7   81.74
  4979.2   82.24  5002.7    82.4  5020.6   82.95 5034.51  83.836  5048.8    84.4
  5053.8   84.22  5071.3   85.24  5081.4   85.46  5101.7   86.84  5122.5   87.42
#Mann= 4 ,-1 , 0
  4746.7     .12       0  4933.3      .1       0  4934.2     .03       0
 5034.51      .1       0
Bank Sta=4934.2,5034.51
XS Rating Curve= 0 ,0
Exp/Cntr=0.3,0.1

Type RM Length L Ch R = 1 ,14974   ,474,474,474
BEGIN DESCRIPTION:
WOODSONS GULLY 28.0
END DESCRIPTION:
XS GIS Cut Line= 3
      3876007.87     10035829.51      3875876.65     10035707.31
      3875830.42     10035514.79
#Sta/Elev= 30
  4821.5   87.18  4841.6   86.07  4848.9   86.43  4884.1    85.1  4898.3   84.32
  4926.6   83.46  4933.5    82.1  4940.3   82.52  4947.6   82.43    4955   83.04
  4961.8   82.12  4969.1      82  4983.3   82.48  4996.6   82.05  5019.9   82.07
  5021.4   81.82  5021.9   81.32  5033.6   81.32  5034.1   81.82  5048.4   82.15
  5056.7   82.97  5079.2   84.11  5089.5   84.23  5098.7    84.9  5103.8   84.89
  5120.3   85.99  5145.8   85.85  5151.2   86.31  5171.8   87.09  5198.8   87.37
#Mann= 4 ,-1 , 0
  4821.5     .12       0  4940.3      .1       0    4955     .03       0
  5056.7      .1       0
Bank Sta=4955,5056.7
XS Rating Curve= 0 ,0
Exp/Cntr=0.3,0.1

Type RM Length L Ch R = 1 ,14500   ,470,470,470
BEGIN DESCRIPTION:
WOODSONS GULLY 27.0
END DESCRIPTION:
XS GIS Cut Line= 3
      3876268.32     10035676.07      3876237.29     10035487.81
      3876122.35     10035368.31
#Sta/Elev= 30
  4809.2   86.33    4820   86.21  4846.3   85.97  4864.9   85.15  4875.1   85.38
  4885.2   84.75  4902.4   84.76  4907.4   84.35  4935.9    84.1    4947   83.28
  4963.5   81.85  5011.3   81.67  5019.1   81.49  5019.6   80.99  5031.3   80.99
  5032.7   81.92  5039.6   81.67  5046.9   81.97  5053.8   83.29  5067.9   83.94
  5075.2   83.92  5082.1   84.72  5089.3   84.69  5096.2   85.35  5103.5   84.89
  5110.4   85.44  5128.4   85.84  5138.7   86.25  5145.9   86.06  5165.8   87.32
#Mann= 5 ,-1 , 0
  4809.2      .1       0    4820     .12       0    4947     .03       0
  5053.8      .1       0  5128.4     .05       0
Bank Sta=4947,5053.8
XS Rating Curve= 0 ,0
Exp/Cntr=0.3,0.1
