--- BELL CREEK.prj (project) ---

Proj Title=BELL CREEK Base Level Engineering
Current Plan=p01
Default Exp/Contr=0.3,0.1
English Units
Geom File=g01
Flow File=f01
Flow File=f02
Plan File=p01
Y Axis Title=Elevation
X Axis Title(PF)=Main Channel Distance
X Axis Title(XS)=Station
BEGIN DESCRIPTION:
BELL CREEK
END DESCRIPTION:
DSS Export Rating Curves= 0
DSS Export Rating Curve Sorted= 0
DSS Export Volume Flow Curves= 0
DXF OffsetX= 0
DXF OffsetY= 0
DXF ScaleX= 1
DXF ScaleY= 10

--- BELL CREEK.p01 (plan) ---

Plan Title=Multiple Run
Short Identifier=Multiple
Geom File=g01
Flow File=f01
Subcritical Flow
K Sum by GR= 0
Std Step Tol= 0.01
Critical Tol= 0.01
Num of Std Step Trials= 20
Max Error Tol= 0.3
Flow Tol Ratio= 0.001
Split Flow NTrial= 30
Split Flow Tol= 0.02
Split Flow Ratio= 0.02
Log Output Level= 0
Friction Slope Method= 1
Unsteady Friction Slope Method= 2
Unsteady Bridges Friction Slope Method= 1
Parabolic Critical Depth
Global Vel Dist=  1 , 1 , 1
Global Log Level= 0
CheckData=True
Encroach Param= -1, 0, 0, 0
BEGIN DESCRIPTION:
Multiple Run
END DESCRIPTION:

--- BELL CREEK.f01 (steady flow) ---

Flow Title=Multiple
Program Version=4.10
Number of Profiles= 7
Profile Names=10-year,25-year,50-year,1pct_min,100-year,1pct_plu,500-year
River Rch & RM=BELL CREEK,Reach-1         ,30500
     266     341     444     191     577    1743    1008
River Rch & RM=BELL CREEK,Reach-1         ,30000
     761    1036    1406     627    1895    5723    3560
River Rch & RM=BELL CREEK,Reach-1         ,22000
     892    1219    1656     739    2232    6741    4192
River Rch & RM=BELL CREEK,Reach-1         ,20249
    2023    2895    4058    1865    5633   17011   11228
River Rch & RM=BELL CREEK,Reach-1         ,20151
    2023    2895    4058    1865    5633   17011   11228
River Rch & RM=BELL CREEK,Reach-1         ,19500
    2023    2895    4058    1865    5633   17011   11228
River Rch & RM=BELL CREEK,Reach-1         ,19071
    2023    2895    4058    1865    5633   17011   11228
River Rch & RM=BELL CREEK,Reach-1         ,18500
    2023    2895    4058    1865    5633   17011   11228
River Rch & RM=BELL CREEK,Reach-1         ,18000
    2023    2895    4058    1865    5633   17011   11228
River Rch & RM=BELL CREEK,Reach-1         ,17500
    2023    2895    4058    1865    5633   17011   11228
River Rch & RM=BELL CREEK,Reach-1         ,15500
    2464    3530    4953    2275    6871   20750   13679
River Rch & RM=BELL CREEK,Reach-1         ,9500
    2443    3471    4843    2211    6676   20161   13125
River Rch & RM=BELL CREEK,Reach-1         ,7000
    2750    3933    5512    2527    7630   23042   15131
River Rch & RM=BELL CREEK,Reach-1         ,4500
    2334    3275    4529    2047    6183   18672   11926
Boundary for River Rch & Prof#=BELL CREEK,Reach-1         , 1
Up Type= 0
Dn Type= 3
Dn Slope=0.005
Boundary for River Rch & Prof#=BELL CREEK,Reach-1         , 2
Up Type= 0
Dn Type= 3
Dn Slope=0.005
Boundary for River Rch & Prof#=BELL CREEK,Reach-1         , 3
Up Type= 0
Dn Type= 3
Dn Slope=0.005
Boundary for River Rch & Prof#=BELL CREEK,Reach-1         , 4
Up Type= 0
Dn Type= 3
Dn Slope=0.005
Boundary for River Rch & Prof#=BELL CREEK,Reach-1         , 5
Up Type= 0
Dn Type= 3
Dn Slope=0.005
Boundary for River Rch & Prof#=BELL CREEK,Reach-1         , 6
Up Type= 0
Dn Type= 3
Dn Slope=0.005
Boundary for River Rch & Prof#=BELL CREEK,Reach-1         , 7
Up Type= 0
Dn Type= 3
Dn Slope=0.005
DSS Import GetInterval= 0
DSS Import GetPeak= 0
DSS Import FillOption= 0

--- BELL CREEK.f02 (steady flow) ---

Flow Title=Orig_BLE_Flow
Program Version=4.10
Number of Profiles= 7
Profile Names=10-year,25-year,50-year,1pct_min,100-year,1pct_plu,500-year
River Rch & RM=BELL CREEK,Reach-1         ,30500
     266     334     386     147     444    1342     586
River Rch & RM=BELL CREEK,Reach-1         ,30000
     761    1016    1223     483    1458    4404    2070
River Rch & RM=BELL CREEK,Reach-1         ,22000
     892    1195    1440     568    1717    5184    2437
River Rch & RM=BELL CREEK,Reach-1         ,20249
    2023    2838    3529    1435    4333   13086    6528
River Rch & RM=BELL CREEK,Reach-1         ,20151
    2023    2838    3529    1435    4333   13086    6528
River Rch & RM=BELL CREEK,Reach-1         ,19500
    2023    2838    3529    1435    4333   13086    6528
River Rch & RM=BELL CREEK,Reach-1         ,19071
    2023    2838    3529    1435    4333   13086    6528
River Rch & RM=BELL CREEK,Reach-1         ,18500
    2023    2838    3529    1435    4333   13086    6528
River Rch & RM=BELL CREEK,Reach-1         ,18000
    2023    2838    3529    1435    4333   13086    6528
River Rch & RM=BELL CREEK,Reach-1         ,17500
    2023    2838    3529    1435    4333   13086    6528
River Rch & RM=BELL CREEK,Reach-1         ,15500
    2464    3461    4307    1750    5285   15960    7953
River Rch & RM=BELL CREEK,Reach-1         ,9500
    2443    3403    4211    1700    5135   15507    7631
River Rch & RM=BELL CREEK,Reach-1         ,7000
    2750    3856    4793    1943    5869   17725    8797
River Rch & RM=BELL CREEK,Reach-1         ,4500
    2334    3211    3938    1575    4756   14363    6934
Boundary for River Rch & Prof#=BELL CREEK,Reach-1         , 1
Up Type= 0
Dn Type= 3
Dn Slope=0.005
Boundary for River Rch & Prof#=BELL CREEK,Reach-1         , 2
Up Type= 0
Dn Type= 3
Dn Slope=0.005
Boundary for River Rch & Prof#=BELL CREEK,Reach-1         , 3
Up Type= 0
Dn Type= 3
Dn Slope=0.005
Boundary for River Rch & Prof#=BELL CREEK,Reach-1         , 4
Up Type= 0
Dn Type= 3
Dn Slope=0.005
Boundary for River Rch & Prof#=BELL CREEK,Reach-1         , 5
Up Type= 0
Dn Type= 3
Dn Slope=0.005
Boundary for River Rch & Prof#=BELL CREEK,Reach-1         , 6
Up Type= 0
Dn Type= 3
Dn Slope=0.005
Boundary for River Rch & Prof#=BELL CREEK,Reach-1         , 7
Up Type= 0
Dn Type= 3
Dn Slope=0.005
DSS Import GetInterval= 0
DSS Import GetPeak= 0
DSS Import FillOption= 0

--- BELL CREEK.g01 (geometry) ---

Geom Title=Existing Conditions
Program Version=4.10

River Reach=BELL CREEK      ,Reach-1
Reach XY= 30
      3811195.05     10150274.62      3810866.57     10149970.71
       3810800.6     10149630.08      3810254.42     10149153.35
      3809818.31     10148891.93      3809036.27     10148814.85
      3809021.43     10148358.08      3808761.79      10148383.6
      3808238.23     10147996.84      3808028.23     10147326.84
      3807188.23     10146676.84      3806698.23     10145856.84
       3806241.8     10145648.65      3806159.86     10145389.59
      3806306.76     10145040.41      3805591.44     10143994.03
      3805179.59     10142855.02      3805186.36     10142159.13
       3805859.4     10141392.05      3805850.15     10139242.02
      3805159.25     10137898.31      3804679.49     10136163.13
      3804656.85     10135469.88      3804187.29     10134529.45
      3803994.17      10133567.4      3803216.24     10132274.62
       3802956.1     10130971.97      3800761.07     10128903.18
       3800149.2      10127537.4      3799909.58     10126201.31

Type RM Length L Ch R = 1 ,30500   ,500,500,500
BEGIN DESCRIPTION:
BELL CREEK 61.0
END DESCRIPTION:
XS GIS Cut Line= 3
      3811681.55     10150134.86      3811160.62     10150245.24
      3810401.58     10150414.12
#Sta/Elev= 30
  4467.5  270.16  4553.1     269  4569.1  270.07  4574.2  268.82  4613.7  270.67
  4618.8  268.77  4663.4  267.98  4668.5  268.62  4675.7  267.42  4726.8  267.66
  4807.3  264.67  4956.3  264.32  4992.6  260.14  4998.9  260.83  5004.1  258.54
  5007.6  258.54  5013.1  262.06  5043.8  263.55  5269.2  263.04  5320.4  263.63
    5331  264.59  5351.1  263.83    5418  264.36  5423.1  265.15  5466.6   264.7
  5494.6  265.19  5510.1  266.63  5535.6  265.69  5576.5  266.02  5777.6  271.35
#Mann= 3 , 0 , 0
  4467.5     .11       0  4956.3     .07       0  5043.8     .11       0
#XS Ineff= 2 , 0
       0  4921.1  264.56    5331       0  264.59
Permanent Ineff=
       F       F
Bank Sta=4956.3,5043.8
XS Rating Curve= 0 ,0
Exp/Cntr=0.3,0.1

Type RM Length L Ch R = 1 ,30000   ,500,500,500
BEGIN DESCRIPTION:
BELL CREEK 60.0
END DESCRIPTION:
XS GIS Cut Line= 3
      3811340.91     10149762.11      3810836.72     10149879.15
      3810317.83     10150261.09
#Sta/Elev= 30
  4482.4  271.41  4548.2  269.59  4670.3   267.4  4817.4  263.39  4916.7  260.11
  4937.1  257.46  4942.3  258.44    4968  258.54  4978.3  258.05  4982.9  257.45
  4983.2  256.95  4986.7  256.95  4986.9  257.45    4990  258.03  5029.1   257.8
  5043.7  259.37  5200.4  260.84  5235.8  262.85  5258.9  263.25  5279.8   264.6
    5309  265.24  5350.8  267.26  5436.4  267.65    5451  268.06    5458  269.06
  5465.7  269.23  5530.5  269.11  5544.9  269.97  5586.8  270.12  5644.3  271.86
#Mann= 4 ,-1 , 0
  4482.4     .11       0  4817.4     .17       0  4916.7     .09       0
  5043.7     .17       0
Bank Sta=4916.7,5043.7
XS Rating Curve= 0 ,0
Exp/Cntr=0.3,0.1

Type RM Length L Ch R = 1 ,29500   ,490,490,490
BEGIN DESCRIPTION:
BELL CREEK 59.0
END DESCRIPTION:
XS GIS Cut Line= 3
      3811154.49     10149302.04      3810574.15     10149564.19
       3810182.7     10150095.94
#Sta/Elev= 30
  4363.2  271.52  4472.4  267.94  4518.7  265.64  4737.7  259.73  4766.3  257.88
  4812.6  257.85  4835.7  256.66  4858.8  257.53  4862.5  255.99  4881.9  256.89
  4887.4  257.76  4897.2  257.25  4933.6  258.53  5002.3  257.63  5045.8  258.64
  5052.4  258.57  5058.6  257.47  5081.7   257.7    5138  259.48    5182  259.96
  5188.2  261.41  5202.8  262.66  5217.5  260.88  5281.7  262.81  5303.1  264.28
  5409.6  265.46    5489  268.76  5539.1  268.78    5589   270.1  5660.3  271.63
#Mann= 4 ,-1 , 0
  4363.2     .11       0  4933.6     .06       0  5045.8     .11       0
    5589     .17       0
Bank Sta=4933.6,5045.8
XS Rating Curve= 0 ,0
Exp/Cntr=0.3,0.1

Type RM Length L Ch R = 1 ,29010   ,510,510,510
BEGIN DESCRIPTION:
BELL CREEK 58.0
END DESCRIPTION:
XS GIS Cut Line= 3
       3810790.5     10148830.31       3810263.1     10149204.73
       3809908.2     10149820.36
#Sta/Elev= 30
  4353.2  272.58  4570.8     266    4738  259.06  4749.1  259.23  4763.9  257.84
  4793.4  257.35  4900.4  252.62  4915.2  252.76  4950.9   251.3  4965.6  249.75
  4971.8  250.92  4980.4  249.92  4986.5  251.83  4998.2  248.78  5001.7  248.78
  5007.3  251.18  5022.6   252.2  5048.9  252.34  5111.2  252.73  5134.3  253.78
  5140.4  253.19  5149.3  253.95  5168.9  253.53  5244.7  255.86  5295.5  257.98
    5521   263.8  5549.8  263.48  5564.1  264.53  5595.7  264.81  5710.6  268.58
#Mann= 7 ,-1 , 0
  4353.2     .11       0    4738     .15       0  4915.2     .09       0
  5022.6     .15       0  5048.9     .17       0  5149.3     .11       0
  5244.7     .17       0
Bank Sta=4915.2,5022.6
XS Rating Curve= 0 ,0
Exp/Cntr=0.3,0.1

Type RM Length L Ch R = 1 ,28500   ,487,487,487
BEGIN DESCRIPTION:
BELL CREEK 57.0
END DESCRIPTION:
XS GIS Cut Line= 3
      3810362.43     10148524.57      3809907.14     10148955.08
      3809722.13     10149717.24
#Sta/Elev= 30
  4373.4  267.63  4402.5  267.56  4437.7  265.29  4451.9  266.11  4459.2  265.39
  4473.3  265.91  4558.3  264.67  4749.2  258.38  4785.8  255.96  4812.7   254.2
  4826.9  254.49    4841  257.54  4847.9   257.2  4855.2  255.39  4862.1  255.26
  4869.4  253.11  4876.2  253.18  4890.4  251.33  4989.5  248.86  4996.1  246.94
  5004.4  246.03  5014.8  247.17  5019.9  249.19  5055.6   249.4  5150.4  248.64
  5170.8  250.14  5192.2   249.4  5201.7  250.82  5275.7  251.38  5784.3  266.27
#Mann= 5 ,-1 , 0
  4373.4     .11       0  4785.8     .17       0  4989.5     .09       0
  5019.9     .15       0  5055.6     .17       0
#XS Ineff= 3 ,-1
  5222.3  5233.9   251.1  5233.9  5270.6  251.31  5270.6    5284  251.66
Permanent Ineff=
       F       F       F
Bank Sta=4989.5,5019.9
XS Rating Curve= 0 ,0
Exp/Cntr=0.3,0.1

Type RM Length L Ch R = 1 ,28013   ,513,513,513
BEGIN DESCRIPTION:
BELL CREEK 56.0
END DESCRIPTION:
XS GIS Cut Line= 3
      3809896.55     10148268.29      3809470.13     10148850.79
      3809427.76     10149656.67
#Sta/Elev= 30
  4278.1  262.86  4315.8  263.24  4501.4  261.16  4616.2  258.88  4672.8  257.11
  4764.9  252.53  4823.4  250.92  4901.2  246.95  4909.1  245.47  4923.7   245.4
  4950.8  243.68  4980.1  243.04    4988  241.05  4992.8  238.85    4993  238.35
  5002.6  238.89  5010.3  241.99  5050.4  243.23  5120.5  243.44    5137  240.33
    5142  240.11  5160.5  242.18  5170.5   240.5  5180.5  239.97  5190.5  243.25
  5220.6  245.62  5240.6  245.54  5420.9  254.01  5601.1  260.98    5807  266.47
#Mann= 4 ,-1 , 0
  4278.1     .11       0  4315.8     .17       0  4980.1     .09       0
  5050.4     .17       0
#XS Ineff= 2 , 0
       0                  5220.6       0  245.62
Permanent Ineff=
       F       F
Bank Sta=4980.1,5050.4
XS Rating Curve= 0 ,0
Exp/Cntr=0.3,0.1

Type RM Length L Ch R = 1 ,27500   ,500,500,500
BEGIN DESCRIPTION:
BELL CREEK 55.0
END DESCRIPTION:
XS GIS Cut Line= 3
      3809675.25     10148116.85      3809031.54     10148805.97
      3808964.81     10149627.17
#Sta/Elev= 30
    4057  261.74  4178.4  260.07  4334.2  256.06  4369.4   254.3  4440.2  252.32
  4525.2  248.17  4539.4  248.18  4596.1  245.05  4617.1  244.61  4638.1  242.54
  4716.3  240.09  4737.3  238.54  4857.4  238.71  4899.9  239.77  4978.1  240.29
  4992.3   238.4  4997.3  234.99  5000.8  234.99  5005.1  237.52  5015.1  240.31
  5045.2  243.05  5103.9  244.39  5135.5  246.34  5217.7  249.15  5264.3  250.99
  5396.4  255.13  5474.6  258.81  5628.1  263.84  5721.3  266.56  5823.9  268.46
#Mann= 7 ,-1 , 0
    4057     .17       0  4978.1     .09       0  5015.1     .17       0
  5217.7     .11       0  5264.3     .17       0  5628.1     .11       0
  5721.3     .17       0
Bank Sta=4978.1,5015.1
XS Rating Curve= 0 ,0
Exp/Cntr=0.3,0.1

Type RM Length L Ch R = 1 ,27000   ,514,514,514
BEGIN DESCRIPTION:
BELL CREEK 54.0
END DESCRIPTION:
XS GIS Cut Line= 4
      3809547.15     10147974.15       3809029.7     10148371.48
      3808883.19     10148742.93      3808792.27     10149622.24
#Sta/Elev= 30
  4347.6  261.34  4395.4  260.53  4422.6  260.91  4495.1   258.6  4501.4  259.14
  4530.5  257.37  4594.8  255.69  4700.8  250.79  4723.5   250.7  4779.7  248.52
  4908.4  240.11  4979.1  237.81  4996.3  232.81  4999.8  232.81  5022.6  236.97
  5095.7  236.24  5214.7  237.92  5225.3  237.51  5246.8  238.79  5287.8  239.04
  5518.1  245.35  5705.5  252.26  5839.8  255.62  6067.8  258.78  6091.6  259.14
  6141.4   260.2  6178.5  261.98  6183.5  261.42  6277.4  263.32  6283.3  262.68
#Mann= 6 ,-1 , 0
  4347.6     .17       0  4979.1     .09       0  5022.6     .17       0
  5705.5     .11       0  6067.8     .17       0  6091.6     .11       0
Bank Sta=4979.1,5022.6
XS Rating Curve= 0 ,0
Exp/Cntr=0.3,0.1

Type RM Length L Ch R = 1 ,26486   ,404,404,404
BEGIN DESCRIPTION:
BELL CREEK 53.0
END DESCRIPTION:
XS GIS Cut Line= 3
      3809340.85     10147834.06      3808623.23     10148291.84
      3807806.12     10148674.34
#Sta/Elev= 30
  4148.8  259.53    4213  258.18  4337.3  252.54  4446.5   249.8  4555.6  245.51
  4634.4  241.28  4662.4  241.01  4743.5  237.52  4858.6  234.74  4958.9   233.3
  4967.8  231.74  4988.9     231  5003.4  229.33  5006.9  229.33    5017   232.3
    5028  232.98  5061.9  233.45  5094.3  232.44  5102.1  233.73  5138.4   233.8
  5160.5  232.35  5182.6  234.15  5250.1  237.61  5289.7  238.32  5295.8  237.89
  5304.1  239.16  5348.2  240.07  5626.5  249.54  5786.4  256.39  5902.2   260.2
#Mann= 4 ,-1 , 0
  4148.8     .17       0  4958.9     .09       0    5028     .17       0
  5289.7     .11       0
Bank Sta=4958.9,5028
XS Rating Curve= 0 ,0
Exp/Cntr=0.3,0.1

Type RM Length L Ch R = 1 ,26082   ,82,82,82
BEGIN DESCRIPTION:
Mapping XS eb4e5b1c
END DESCRIPTION:
XS GIS Cut Line= 3
      3809205.37     10147799.43      3808343.71     10148094.65
      3807693.32     10148365.85
#Sta/Elev= 30
    4091   257.1  4238.3  251.81  4358.1  250.41  4571.8  241.85  4680.3  235.49
  4728.2  235.11  4733.5  233.68  4754.2  234.22  4816.8  232.49  4822.1  231.37
  4848.1  232.26  4853.4  230.79  4879.3  231.71  4884.6  230.33  4910.6  231.93
  4915.9  230.07  4923.5  229.83  4973.2   230.7  4978.5  229.53  5004.1  229.17
  5007.8  226.49  5040.7  230.68  5157.9  235.33  5192.6  238.25    5211  236.92
  5216.4  238.45  5240.2  240.23  5298.3  242.67  5529.4  251.91  5706.5  257.27
#Mann= 4 ,-1 , 0
    4091     .17       0  4973.2     .09       0  5040.7     .17       0
  5298.3     .11       0
#XS Ineff= 2 , 0
       0  4754.2  234.22               0
Permanent Ineff=
       F       F
Bank Sta=4973.2,5040.7
XS Rating Curve= 0 ,0
Exp/Cntr=0.3,0.1

Type RM Length L Ch R = 1 ,26000   ,500,500,500
BEGIN DESCRIPTION:
BELL CREEK 52.0
END DESCRIPTION:
XS GIS Cut Line= 3
      3809183.76     10147717.83      3808301.34     10148029.95
      3807641.68     10148298.17
#Sta/Elev= 30
    4064  257.69  4447.7  248.59    4566  242.19  4571.3  240.01  4596.9  240.33
  4627.8  239.05  4633.1  237.53  4833.5  230.81  4869.8  231.02  4895.4  228.97
  4900.7  230.67  4924.5  227.96  4988.1  230.47  5004.6  228.72  5012.7  230.53
  5090.1  229.81  5149.2  235.69  5202.8   238.2  5226.8  237.57  5273.6  242.23
  5280.4  244.81  5285.8  243.16  5304.5   247.7  5309.9  246.39  5322.1  247.17
  5333.9   243.6  5339.3  245.62    5358  242.21  5403.2  246.68  5712.1  255.96
#Mann= 4 ,-1 , 0
    4064     .17       0  4988.1     .09       0  5012.7     .17       0
  5322.1     .11       0
Bank Sta=4988.1,5012.7
XS Rating Curve= 0 ,0
Exp/Cntr=0.3,0.1

Type RM Length L Ch R = 1 ,25500   ,592,592,592
BEGIN DESCRIPTION:
BELL CREEK 51.0
END DESCRIPTION:
XS GIS Cut Line= 3
       3809045.7     10147472.94      3808138.23     10147651.66
      3807538.78     10148184.75
#Sta/Elev= 30
  4075.1  257.39  4113.7  257.73  4197.6  255.05    4403  252.19  4490.8   250.1
  4633.5  243.24  4711.1  238.26  4745.6   237.5  4762.5  235.85  4767.6  236.57
  4776.2  235.41  4916.5  227.65  4939.2  227.49    4980  228.75  4988.4  226.18
  5013.9  228.71  5049.6   227.6  5084.7  228.01  5134.3  230.87  5162.5   230.6
  5184.2   232.5  5205.1  232.87  5339.7  239.98  5368.2  240.38  5474.4  245.11
  5509.5   245.5  5566.3  248.76  5573.9  248.12  5610.8  249.82  5802.2  255.81
#Mann= 4 ,-1 , 0
  4075.1     .17       0    4980     .09       0  5013.9     .17       0
  5610.8     .11       0
Bank Sta=4980,5013.9
XS Rating Curve= 0 ,0
Exp/Cntr=0.3,0.1

Type RM Length L Ch R = 1 ,24908   ,393,393,393
BEGIN DESCRIPTION:
BELL CREEK 50.0
END DESCRIPTION:
XS GIS Cut Line= 3
      3808927.64     10147290.06      3808018.23     10147316.84
      3807441.55     10148088.71
#Sta/Elev= 30
  4090.2  254.16    4120  254.79    4210   252.4  4380.1  251.22  4520.2  248.71
  4620.2  244.01  4629.6   244.4  4650.2  242.72  4660.2  243.03  4670.2  241.59
  4720.3  238.34  4790.3  235.85  4870.3  230.99  4960.4  226.93  4990.4  224.83
  5004.5  225.05  5008.5   223.6    5012   223.6  5017.8  226.31  5031.1  226.87
  5060.3  225.95  5131.1  225.77  5160.3  227.45  5231.2  228.99  5304.2  232.63
  5525.1  239.63  5725.2  247.89  5819.5  250.36    5904  251.77  5963.5  254.32
#Mann= 4 ,-1 , 0
  4090.2     .17       0  4960.4     .09       0  5031.1     .17       0
  5819.5     .11       0
Bank Sta=4960.4,5031.1
XS Rating Curve= 0 ,0
Exp/Cntr=0.3,0.1

Type RM Length L Ch R = 1 ,24515   ,480,480,480
BEGIN DESCRIPTION:
BELL CREEK 49.0
END DESCRIPTION:
XS GIS Cut Line= 3
      3808261.68     10146777.62       3807731.4     10147116.84
      3807346.75     10147995.43
#Sta/Elev= 30
  4370.5  244.68    4529  243.13    4654  239.27  4686.4   237.5  4722.7  236.82
  4859.3   227.6  4889.3  226.43  4904.5  226.99    4933  224.95  4977.3  224.22
  4990.6  220.71  4994.1  220.71  4998.4  223.17  5015.5  224.18  5044.5  224.19
  5059.2  223.26  5067.9  224.46  5096.8  224.18  5157.4  225.39  5274.3  229.73
  5310.3   231.8  5353.9  232.35  5370.4   233.8  5504.2  239.37  5623.5  242.76
    5684  244.55  5719.6  244.75  5818.5  247.63  5870.8  247.71  5959.1  250.13
#Mann= 9 ,-1 , 0
  4370.5     .17       0    4654     .11       0  4859.3     .15       0
  4977.3     .09       0  5015.5     .15       0  5274.3     .17       0
  5504.2     .11       0  5623.5     .17       0    5684     .11       0
Bank Sta=4977.3,5015.5
XS Rating Curve= 0 ,0
Exp/Cntr=0.3,0.1

Type RM Length L Ch R = 1 ,24035   ,552,552,552
BEGIN DESCRIPTION:
BELL CREEK 48.0
END DESCRIPTION:
XS GIS Cut Line= 3
      3808252.32     10146737.47      3807488.23     10146816.84
      3806598.79     10147423.62
#Sta/Elev= 30
  4231.8  244.14  4266.5  243.89  4286.6  243.06  4346.9  243.06  4555.6   239.2
  4648.5  238.15    4749  235.55  4789.3  232.98  4819.4  229.53  4854.4  227.43
  4909.9  223.97  4993.9  222.12  4995.9  220.23  5011.4  220.85  5017.5  222.35
  5047.3  221.29  5091.8  222.17  5133.6  222.85  5169.9  222.36    5197  223.78
  5218.4  223.04  5226.9  223.68  5241.8  223.31  5319.6  224.78  5478.2  229.47
  5693.6  237.27  5923.9  243.16  5938.9  244.29  5974.8  244.24  6076.7  247.86
#Mann= 6 ,-1 , 0
  4231.8     .17       0  4555.6     .11       0  4854.4     .15       0
  4993.9     .09       0  5017.5     .15       0  5091.8     .11       0
#XS Ineff= 2 , 0
       0                  5313.6       0  224.86
Permanent Ineff=
       F       F
Bank Sta=4993.9,5017.5
XS Rating Curve= 0 ,0
Exp/Cntr=0.3,0.1

Type RM Length L Ch R = 1 ,23483   ,483,483,483
BEGIN DESCRIPTION:
BELL CREEK 47.0
END DESCRIPTION:
XS GIS Cut Line= 3
      3808277.09     10146697.28      3807118.23     10146576.84
      3806540.01     10147355.67
#Sta/Elev= 30
  3834.9  243.27  3924.6  242.72  4179.4  238.88  4206.1  237.88  4232.4  238.31
  4447.4  235.27    4558  230.49  4654.7  225.15    4749  222.24  4769.1  222.37
  4779.2  221.03  4799.3  220.13    4930  218.95  4970.2  219.48  4980.3  218.86
  4990.3   216.6  4995.9  213.85  5004.5  214.35  5010.3  217.91  5024.9  219.65
  5061.9   219.2  5095.8  219.85  5117.4  221.45  5195.9  224.42    5390  229.61
    5511  233.84  5732.1  239.36  5876.1   244.4  5911.6  246.41    5970  247.71
#Mann= 6 ,-1 , 0
  3834.9     .17       0  4179.4     .11       0  4654.7     .15       0
  4970.2     .09       0  5024.9     .15       0  5061.9     .11       0
Bank Sta=4970.2,5024.9
XS Rating Curve= 0 ,0
Exp/Cntr=0.3,0.1

Type RM Length L Ch R = 1 ,23000   ,479,479,479
BEGIN DESCRIPTION:
BELL CREEK 46.0
END DESCRIPTION:
XS GIS Cut Line= 3
      3807467.29     10146199.66      3806915.62     10146194.23
      3806122.81     10146712.72
#Sta/Elev= 30
  4448.3  231.24  4507.7  230.11  4607.7  231.44  4627.7  230.02  4697.8  228.94
  4797.8   225.5  4885.2   220.2  4947.8  217.29  4957.8   215.5  4967.8  216.04
  4994.6  212.74  5003.3  213.34  5009.3  215.68  5018.4  217.11  5075.7  217.09
  5117.9  214.89  5150.8  216.71  5407.4  223.46  5531.1  223.69  5546.2  224.18
  5552.2  225.35  5567.3  223.62  5573.3  224.72  5582.4  222.76  5588.4  222.83
  5603.5  225.57  5862.8  235.05  5883.9  236.78  5935.2  237.82  5947.3  238.97
#Mann= 5 ,-1 , 0
  4448.3     .11       0  4885.2     .15       0  4947.8     .09       0
  5018.4     .15       0  5150.8     .11       0
Bank Sta=4947.8,5018.4
XS Rating Curve= 0 ,0
Exp/Cntr=0.3,0.1

Type RM Length L Ch R = 1 ,22521   ,521,521,521
BEGIN DESCRIPTION:
BELL CREEK 45.0
END DESCRIPTION:
XS GIS Cut Line= 3
      3807331.33     10146008.03      3806698.23     10145856.84
      3806005.33     10146539.65
#Sta/Elev= 30
  4349.1   229.2  4414.4  228.68    4476  230.26  4537.7  228.98  4568.1  229.75
  4746.8  226.86  4788.8  225.84    4815  223.92  4915.6  217.79  4962.3  216.61
 4966.88  214.68  4979.8  211.33  4990.1  209.93  4995.9  207.73  5010.3  209.13
  5017.4  212.15  5024.5  212.16  5031.5  213.69  5038.6  212.02  5045.7  212.02
  5052.8  210.67  5066.9  210.47  5073.9  212.94  5088.1  214.67  5151.8  214.51
  5165.9  213.13  5187.1  215.55  5264.9  217.64  5342.7  217.76  5972.8   238.3
#Mann= 5 ,-1 , 0
  4349.1     .11       0    4815     .17       0  4915.6     .15       0
 4966.88     .09       0  5088.1     .11       0
Bank Sta=4966.88,5088.1
XS Rating Curve= 0 ,0
Exp/Cntr=0.3,0.1

Type RM Length L Ch R = 1 ,22000   ,430,430,430
BEGIN DESCRIPTION:
BELL CREEK 44.0
END DESCRIPTION:
XS GIS Cut Line= 4
      3807340.53     10145949.29      3806472.72      10145686.6
      3806306.21     10145704.82      3805943.51     10146462.37
#Sta/Elev= 30
  3925.8  227.32  4077.5  227.26  4168.9  229.13  4273.4  227.98  4389.6  226.14
  4455.4  223.51  4488.4  220.95  4555.4  220.14  4663.5  214.18  4711.1  214.57
    4813  213.62  4867.6  213.34  4887.7  211.61  4916.2  213.31  4921.2  211.12
  4927.9  212.92    4948   212.8  4968.2  210.95  4978.2  208.94  4986.5  205.13
    5000  207.56  5010.1   212.1    5018  212.69  5287.7     222  5633.2  232.26
  5678.5  232.63  5701.2  234.49  5729.4  234.02  5820.1  237.21  5839.9  236.87
#Mann= 6 ,-1 , 0
  3925.8     .11       0  4555.4     .15       0  4711.1     .17       0
    4813     .11       0    4948     .06       0    5018     .11       0
#XS Ineff= 2 ,-1
  4701.8  4649.5  214.67    4754  4701.8  214.29
Permanent Ineff=
       F       F
Bank Sta=4948,5018
XS Rating Curve= 0 ,0
Exp/Cntr=0.3,0.1

Type RM Length L Ch R = 1 ,21570   ,386,386,386
BEGIN DESCRIPTION:
BELL CREEK 43.0
END DESCRIPTION:
XS GIS Cut Line= 3
      3807359.11     10145902.93      3806174.77     10145341.89
      3805452.42     10145414.55
#Sta/Elev= 30
  3689.5  226.56  3916.7  225.92  4053.2  227.33  4365.9  224.75  4426.9  222.65
  4488.2  219.63  4546.9  217.05  4748.6  211.41  4888.1  209.24  4908.1  207.51
  4916.9  209.34  4922.4   208.3  4930.2   209.9  4974.5  210.62  5005.2  204.14
    5017  207.17  5036.9     208  5047.2  210.52  5157.7  212.27  5197.9  218.72
    5208  218.75    5218  216.15  5264.4  216.21  5337.6  218.77  5378.8  217.36
  5398.9  218.25  5437.8  224.72  5442.8  223.85  5459.2  225.83    5726  232.78
#Mann= 9 ,-1 , 0
  3689.5     .11       0  4426.9     .17       0  4488.2     .11       0
  4546.9     .17       0  4748.6     .15       0  4888.1     .17       0
  4974.5     .09       0  5047.2     .17       0  5264.4     .11       0
#XS Ineff= 2 , 0
       0  4706.6   212.1  5127.6       0   212.3
Permanent Ineff=
       F       F
Bank Sta=4974.5,5047.2
XS Rating Curve= 0 ,0
Exp/Cntr=0.3,0.1

Type RM Length L Ch R = 1 ,21184   ,337,337,337
BEGIN DESCRIPTION:
Mapping XS aeda876c
END DESCRIPTION:
XS GIS Cut Line= 3
      3807371.22     10145875.44      3806306.76     10145040.41
      3805441.74     10145343.83
#Sta/Elev= 30
  3647.1  226.23  4108.9  225.52  4165.3  224.51  4357.9  224.06    4629  220.12
  4699.6  217.95  4827.9  211.48  4912.9  210.66  4962.6  208.36  4970.7  204.78
  4977.1  208.09  4985.2  205.62  4991.5   207.9  4996.1  205.03  5002.1  205.03
  5007.5  200.64  5011.3  200.64  5030.6  208.26  5046.9  209.27  5072.6  207.82
  5157.8  208.82  5315.4  212.09  5413.7  215.91  5439.4  219.49  5486.3  222.51
  5496.1   222.6  5501.4  220.86  5518.1  221.12  5719.5  228.94  5916.7  233.45
#Mann= 3 , 0 , 0
  3647.1     .11       0  4962.6     .09       0  5030.6     .11       0
#XS Ineff= 2 , 0
       0  4912.9  210.66               0
Permanent Ineff=
       F       F
Bank Sta=4962.6,5030.6
XS Rating Curve= 0 ,0
Exp/Cntr=0.3,0.1

Type RM Length L Ch R = 1 ,20847   ,338,338,338
BEGIN DESCRIPTION:
BELL CREEK 42.0
END DESCRIPTION:
XS GIS Cut Line= 4
       3807386.9     10145865.81      3806601.93     10144764.27
      3806109.18     10144769.85      3805424.29     10145281.65
#Sta/Elev= 30
  3154.6  226.14  3199.7  225.99    3244   223.9    3330  227.36  3386.6  225.31
  3393.7  223.77  3466.5  225.63  3659.5   222.1  3766.5  222.47  3816.9   220.9
  4219.4  218.21  4495.9  216.86  4582.3  214.98  4687.5  213.92  4731.3   213.4
  4791.3   210.3  4971.3  207.52  4981.3  206.83  4996.3   201.1    5004   201.6
  5015.4  206.69  5023.7  207.77  5044.6  206.89  5165.5  208.02  5323.9  212.01
  5394.8  216.64  5480.2  219.89  5494.8  218.94  5688.3  229.22    5855  233.15
#Mann= 7 ,-1 , 0
  3154.6     .11       0  4219.4     .17       0  4495.9     .11       0
  4582.3    .125       0  4687.5     .11       0  4971.3     .06       0
  5023.7     .11       0
Bank Sta=4971.3,5023.7
XS Rating Curve= 0 ,0
Exp/Cntr=0.3,0.1

Type RM Length L Ch R = 1 ,20509   ,260,260,260
BEGIN DESCRIPTION:
Mapping XS 3d0ebc16
END DESCRIPTION:
XS GIS Cut Line= 4
        3807399.     10145859.81      3806681.57      10144636.3
      3805921.13     10144494.41      3805237.75     10144927.02
#Sta/Elev= 30
  2808.1  226.27  2887.8  223.67  2955.1  227.41    2998  227.64  3056.7  224.05
    3108  223.67  3136.8  225.11  3312.7  221.92  3547.2  221.89  3823.9  217.69
  4060.5  218.42  4377.8  215.53  4577.1  215.11    4688     213  4810.1  207.76
  4972.8  206.26  4989.5     204  4994.6  204.78  4997.2  202.62    5001  202.62
  5006.4  205.08  5015.7  203.68  5021.7  205.74  5027.6  204.42    5037  205.73
  5194.6  206.66  5334.5  209.74  5392.1  211.68  5616.7  224.96  5808.8  230.51
#Mann= 7 ,-1 , 0
  2808.1     .11       0  3823.9     .17       0  4060.5     .11       0
  4377.8    .125       0  4577.1     .11       0  4972.8     .06       0
    5037     .11       0
Bank Sta=4972.8,5037
XS Rating Curve= 0 ,0
Exp/Cntr=0.3,0.1

Type RM Length L Ch R = 1 ,20249   ,98,98,98
BEGIN DESCRIPTION:
BELL CREEK 41.0
END DESCRIPTION:
XS GIS Cut Line= 4
      3807295.17     10143956.98      3806014.82     10144223.33
      3805779.87     10144278.93      3805197.01     10144426.29
#Sta/Elev= 30
  3450.8  217.74    3690   209.7  3805.6  210.25  3885.2  207.69  4280.8  205.56
  4295.8  206.97  4325.7  201.66  4346.9  203.95  4375.8   203.6  4387.8  206.23
  4499.7  205.34  4520.5  204.81  4571.1  208.42  4616.5  205.05  4626.3  207.04
  4671.2  204.87  4676.3  206.92  4765.5  204.41  4770.7  206.36  4812.9  204.35
  4902.6  205.12  4944.9  204.41  4979.1  199.99  5012.4  202.65  5022.7  201.36
  5028.5  203.46  5033.7  202.13  5069.5  205.81  5310.5  208.44  5601.2  219.69
#Mann= 5 ,-1 , 0
  3450.8     .11       0  4499.7    .125       0  4616.5     .11       0
  4902.6     .06       0  5069.5     .11       0
#XS Ineff= 4 ,-1
  4571.1  3840.2  208.42  4770.7  4571.1  206.36  5115.7  5151.6  206.08
  5151.6  5192.6  206.85
Permanent Ineff=
       F       F       F       F
Bank Sta=4902.6,5069.5
XS Rating Curve= 0 ,0
Exp/Cntr=0.3,0.1

Type RM Length L Ch R = 1 ,20151   ,651,651,651
BEGIN DESCRIPTION:
BELL CREEK 40.0
END DESCRIPTION:
XS GIS Cut Line= 3
      3807178.03      10143855.4      3805730.63     10144194.95
      3805157.35     10144309.98
#Sta/Elev= 30
  3513.3  218.93  3538.5  218.27  3607.4  214.51  3720.8  211.95  3842.2  208.75
  4160.6  205.97  4301.8  207.78  4349.4  201.06  4386.6  201.68  4396.9  205.01
  4434.2  207.04  4633.1   206.2  4756.3  208.22  4951.5     205    4964  203.42
    4972  200.38  5010.6  199.82  5023.2  202.45  5057.7  204.74  5072.1  204.73
  5103.5  205.71    5115  208.49  5145.6  208.56  5154.5  206.78  5227.9     210
  5261.4  208.39  5312.3  212.43  5363.2  211.42  5579.2  222.31  5584.7  222.52
#Mann= 8 ,-1 , 0
  3513.3     .11       0  3538.5    .125       0  3720.8     .11       0
  4951.5     .07       0  5057.7     .11       0  5072.1    .125       0
  5227.9     .11       0  5579.2    .125       0
#XS Ineff= 2 , 0
       0  4789.1  207.97  5135.4       0   208.9
Permanent Ineff=
       T       F
Bank Sta=4951.5,5057.7
XS Rating Curve= 0 ,0
Exp/Cntr=0.3,0.1

Type RM Length L Ch R = 1 ,19500   ,429,429,429
BEGIN DESCRIPTION:
BELL CREEK 39.0
END DESCRIPTION:
XS GIS Cut Line= 3
       3806964.7     10143390.29      3805472.11     10143608.07
      3804864.09     10143936.59
#Sta/Elev= 30
  3491.6  220.65  3538.9  218.57  3667.7  218.37  3761.3  216.26  3807.7  218.29
  4017.7  215.56  4083.7  216.31    4184  215.36  4227.7  214.83  4286.8  210.95
  4337.3  201.63  4347.4     201  4429.8  200.96  4430.2  200.46  4435.6  200.96
  4455.5  201.48  4529.3  202.12  4559.6  205.29  4579.9  201.05  4600.1     201
  4637.6  204.67  4759.4  205.67  4812.3  205.48  4917.7  204.12  4943.7     201
  5041.2     201    5073  205.55  5358.1  210.28  5478.1  217.54  5691.1  225.69
#Mann= 9 ,-1 , 0
  3491.6     .11       0  4083.7     .15       0    4184     .17       0
  4429.8     .11       0  4435.6     .17       0  4455.5     .11       0
  4759.4    .125       0  4812.3     .07       0    5073     .11       0
#XS Ineff= 2 , 0
       0  4782.7  205.94  5095.5       0   206.1
Permanent Ineff=
       T       F
Bank Sta=4812.3,5073
XS Rating Curve= 0 ,0
Exp/Cntr=0.3,0.1

Type RM Length L Ch R = 1 ,19071   ,571,571,571
BEGIN DESCRIPTION:
BELL CREEK 38.0
END DESCRIPTION:
XS GIS Cut Line= 3
      3806968.75      10143353.8      3805308.37     10143211.03
      3804510.89     10143263.36
#Sta/Elev= 30
  3333.5  221.06  3565.2  217.44  3777.5   216.4  3826.2  217.72    3919  215.57
  4137.4  210.01  4215.2  210.32  4287.9  209.88  4367.3  205.04  4408.3  201.06
    4546  200.54  4546.4  200.04  4551.8  200.54  4659.3  200.98  4669.3  203.48
  4708.8     201  4739.6     201  4769.7  205.11  4906.2  205.49  4938.2     201
  5050.6  201.48  5081.3  205.36  5271.1  206.86  5321.2  210.99  5391.4  211.02
  5441.5  215.29  5541.7  219.44  5631.9  221.37  5712.1  220.72  5799.2  224.23
#Mann= 9 ,-1 , 0
  3333.5     .11       0    3919     .17       0  4215.2     .11       0
  4367.3     .15       0    4546     .12       0  4551.8     .15       0
  4708.8    .125       0  4906.2     .07       0  5081.3     .11       0
#XS Ineff= 2 , 0
       0  4900.2  205.97  5180.9       0  205.92
Permanent Ineff=
       T       F
Bank Sta=4906.2,5081.3
XS Rating Curve= 0 ,0
Exp/Cntr=0.3,0.1

Type RM Length L Ch R = 1 ,18500   ,500,500,500
BEGIN DESCRIPTION:
BELL CREEK 37.0
END DESCRIPTION:
XS GIS Cut Line= 3
      3806984.41     10143328.47       3805177.3     10142663.99
      3804521.18     10142425.27
#Sta/Elev= 30
  3074.6  220.95  3082.9  220.84  3305.3  217.84  3600.7  217.04  3678.2  215.78
  3699.6  216.62  3731.5  215.59  3997.9  214.03  4183.5  209.29  4189.7  208.16
  4239.1  206.71    4300  206.41  4330.5  205.06  4349.5  203.11  4355.7     201
  4534.4     201  4583.4  202.65  4638.1     201  4658.5     201  4667.6  202.63
  4775.7  204.44  4914.2   203.9  4924.8  202.58  4930.6  200.23  5049.9  200.79
  5063.3  203.03  5085.8  203.93  5236.8  206.04  5425.1   208.2  5698.2  216.77
#Mann= 8 ,-1 , 0
  3074.6    .125       0  3082.9    .125       0  4534.4     .15       0
  4638.1     .11       0  4667.6    .125       0  4914.2     .09       0
  5085.8     .15       0  5236.8     .11       0
#XS Ineff= 2 , 0
       0  4330.5  205.06               0
Permanent Ineff=
       F       F
Bank Sta=4914.2,5085.8
XS Rating Curve= 0 ,0
Exp/Cntr=0.3,0.1

Type RM Length L Ch R = 1 ,18000   ,500,500,500
BEGIN DESCRIPTION:
BELL CREEK 36.0
END DESCRIPTION:
XS GIS Cut Line= 3
       3806993.8     10143304.06      3805181.92     10142173.25
      3804452.23     10141999.89
#Sta/Elev= 30
  2864.2  221.44  3095.2  217.91  3319.4  217.76    3350  216.68  3575.4  214.68
  3625.6  213.12  3669.7  214.11  3696.9  212.94  3742.9  213.05    3895  210.58
  3952.8   208.6  3989.4  209.23    4105  206.12    4184  206.23  4214.7  203.38
  4220.6  204.37  4272.5  202.67  4285.7  204.64  4299.6  203.69  4309.1  201.36
    4315  201.09  4424.7  200.95  4471.8   199.7  4482.5     201  5127.5  200.67
  5137.8  201.44  5148.1  203.53  5415.3  208.69  5631.2  216.39    5750  222.07
#Mann= 3 , 0 , 0
  2864.2     .12       0  4299.6     .07       0  5148.1     .12       0
Bank Sta=4299.6,5148.1
XS Rating Curve= 0 ,0
Exp/Cntr=0.3,0.1

Type RM Length L Ch R = 1 ,17500   ,500,500,500
BEGIN DESCRIPTION:
BELL CREEK 35.0
END DESCRIPTION:
XS GIS Cut Line= 3
       3807004.5      10143294.3       3805507.5     10141814.71
      3804036.72     10141560.45
#Sta/Elev= 30
  2895.2  221.64  3602.2  213.54  3800.2  213.33  3814.4  216.64  3828.5  213.61
  3856.8  212.53  4047.7  211.09  4436.7  203.66    4465     201  4592.2     201
  4601.9  199.66  4613.4     201  5669.4  200.74  5695.6  203.16  5700.7   201.2
  5730.3   203.8  5750.3  206.17  5755.4  204.91  5770.9  205.55  5791.2  209.23
  5810.1   210.6  5815.2  207.66  5821.7  208.96  5852.1  208.73  5892.7  213.72
  6049.3     217  6126.1  221.15  6163.8  220.26  6338.2   227.7  6492.6  231.29
#Mann= 3 , 0 , 0
  2895.2     .11       0  4436.7     .06       0  5730.3     .11       0
#XS Ineff= 2 , 0
       0                  5750.3       0  206.17
Permanent Ineff=
       F       F
Bank Sta=4436.7,5730.3
XS Rating Curve= 0 ,0
Exp/Cntr=0.3,0.1

Type RM Length L Ch R = 1 ,17000   ,500,500,500
BEGIN DESCRIPTION:
BELL CREEK 34.0
END DESCRIPTION:
XS GIS Cut Line= 3
      3807597.99     10142156.64      3805830.36     10141446.37
      3803957.15     10141186.82
#Sta/Elev= 30
    3095  243.46  3224.5  239.62  3289.4  235.12  3396.9  230.78    3703  221.77
  4021.3  211.42    4126   209.3  4251.8  206.72  4353.9  202.17  4359.3  203.43
  4362.5  200.21  4628.1  203.43  4652.3  202.78  4657.8     201  5608.3     201
 5621.21  203.38  5628.5  205.23  5668.8   207.8  5810.2  212.67  5981.8  215.76
  6073.7  215.11  6123.6   214.9  6433.8  215.36  6596.9  214.55    6638  215.31
  6648.1  219.16  6658.2  220.51    6781  225.36  6809.6  226.27  6891.1   234.8
#Mann= 11 ,-1 , 0
    3095     .11       0    3703     .17       0  4021.3     .11       0
    4126     .15       0  4628.1     .06       0 5621.21    .125       0
  6073.7     .11       0  6123.6    .125       0  6433.8     .11       0
  6596.9    .125       0    6781     .11       0
Bank Sta=4628.1,5621.21
XS Rating Curve= 0 ,0
Exp/Cntr=0.3,0.1

Type RM Length L Ch R = 1 ,16500   ,500,500,500
BEGIN DESCRIPTION:
BELL CREEK 33.0
END DESCRIPTION:
XS GIS Cut Line= 3
      3807613.84     10142085.07      3805876.54     10140954.28
      3803702.79     10140789.36
#Sta/Elev= 30
  2927.1  241.85  3216.6  229.05  3289.1  228.61  3439.9  222.11  3888.8  212.47
  4155.4  204.01  4262.8  203.44  4315.4  203.12  4342.5     201  4466.3     201
  4487.4  203.77  4517.6  203.47  4553.9     201  5626.1  200.45  5650.6   203.4
  5720.8  212.35    5811  213.38  5861.2   219.2  5898.9  213.06  5980.1  214.12
  6078.8  214.89  6593.3  215.24  6813.9  217.17  6822.9  219.65  6827.9   218.7
    6854  222.38  6934.2  225.65  6994.4   230.6  7090.4  235.52    7180  233.32
#Mann= 6 ,-1 , 0
  2927.1     .11       0  4262.8     .15       0  4517.6     .06       0
  5650.6     .11       0  5980.1     .15       0  6078.8     .11       0
Bank Sta=4517.6,5650.6
XS Rating Curve= 0 ,0
Exp/Cntr=0.3,0.1

Type RM Length L Ch R = 1 ,16000   ,500,500,500
BEGIN DESCRIPTION:
BELL CREEK 32.0
END DESCRIPTION:
XS GIS Cut Line= 3
      3807868.23     10140757.56      3805895.65     10140454.64
      3803670.99     10140646.27
#Sta/Elev= 30
  3004.3  229.44  3510.5  227.04  3763.5  220.39  3834.3  216.63  4228.9  207.24
  4350.3  206.07  4370.5  204.23  4497.1   200.5  5640.2     201  5715.6  204.42
  5901.1  207.58  5931.2  210.86    5987  209.26  6021.6  208.41    6061  211.92
  6121.9  212.81  6322.7  212.58  6423.1  215.71  6885.4  215.93  6914.9  217.64
  6965.1  226.91  7015.2  230.51  7035.3   233.9  7065.4  243.43  7075.5   243.7
  7095.5  243.11  7135.7  234.05  7155.8  234.26  7175.8  231.72  7232.9  231.75
#Mann= 4 ,-1 , 0
  3004.3     .11       0  4370.5     .06       0  5715.6     .15       0
    5987     .11       0
Bank Sta=4370.5,5715.6
XS Rating Curve= 0 ,0
Exp/Cntr=0.3,0.1

Type RM Length L Ch R = 1 ,15500   ,500,500,500
BEGIN DESCRIPTION:
BELL CREEK 31.0
END DESCRIPTION:
XS GIS Cut Line= 3
       3807939.8     10140654.22      3805849.91     10139961.51
      3803575.64     10140455.48
#Sta/Elev= 30
  2798.3  228.71  2888.8   226.5  2978.6  227.92  3015.6   226.4  3274.4  223.75
  3379.8  224.91  3411.4  222.99  3516.7  220.95  3559.7  221.31    3601  218.97
    3738  217.16  3769.6  215.31  3876.6  213.09  3934.8  210.08  4130.2  205.42
  4383.7  202.82  4391.1  202.68  4395.2   200.5  6803.1     201    6810  205.54
  6815.2  208.82  6844.1  216.39  6864.5  220.16  7001.5  221.54    7018  226.22
  7045.5  229.16  7138.7  230.84  7222.7  234.27  7236.9   232.7  7327.3  232.21
#Mann= 3 , 0 , 0
  2798.3     .11       0  4130.2     .06       0    6810     .11       0
#XS Ineff= 2 , 0
       0    4257  204.52               0
Permanent Ineff=
       F       F
Bank Sta=4130.2,6810
XS Rating Curve= 0 ,0
Exp/Cntr=0.3,0.1

Type RM Length L Ch R = 1 ,15000   ,500,500,500
BEGIN DESCRIPTION:
BELL CREEK 30.0
END DESCRIPTION:
XS GIS Cut Line= 3
      3807780.84     10138181.96      3805850.16     10139461.51
      3803401.82     10140089.54
#Sta/Elev= 30
  2683.8  243.56  2764.5  241.92  2779.6  239.65  2929.9  231.45  2987.3  223.51
  3110.4  213.16  3248.8  207.26  3275.9  204.53  3299.2  205.69  3399.2  204.59
  3465.4  205.81  3564.6  203.78  3594.7  204.86  3651.9  203.18  3754.2  202.11
  3760.5   200.5  7015.5     201  7025.7  201.25  7030.8  203.14  7087.8  221.44
  7098.1  223.44  7107.2  223.46  7112.4  225.47  7129.1  224.37  7201.3  224.66
  7242.6  227.78  7376.8  233.23  7428.2  231.79  7490.4  232.03  7527.6  235.57
#Mann= 3 , 0 , 0
  2683.8     .11       0  3651.9     .06       0  7030.8     .11       0
#XS Ineff= 2 ,-1
  3537.6  3263.2  205.08  3594.7  3537.6  204.86
Permanent Ineff=
       F       F
Bank Sta=3651.9,7030.8
XS Rating Curve= 0 ,0
Exp/Cntr=0.3,0.1

Type RM Length L Ch R = 1 ,14500   ,500,500,500
BEGIN DESCRIPTION:
BELL CREEK 29.0
END DESCRIPTION:
XS GIS Cut Line= 3
      3807757.02     10138094.52      3805724.65     10138991.73
      3803211.36      10139787.3
#Sta/Elev= 30
  2778.4  241.83  3008.8  231.48  3328.3  208.65  3374.9  212.98  3577.8  217.05
  3821.8  205.68  3960.6   200.4  6272.3     201  6476.6  205.74  6600.6  208.42
  6605.8  210.88  6632.9  209.15  6638.1  211.68  6702.7  210.16  6716.8  214.85
    6735  213.32  6740.3   217.4  6767.3  213.65  6772.6  216.53  6837.2  217.99
  6853.2  213.38  6869.5  213.34    6907  216.76  6934.1  214.61  6939.3   217.4
  7369.7  229.43  7429.1  229.91  7504.2  225.27  7536.5   229.8  7636.2  230.08
#Mann= 3 , 0 , 0
  2778.4     .11       0  3821.8     .06       0  6476.6     .11       0
#XS Ineff= 2 ,-1
  6406.8  6444.3  204.77  6444.3  6476.6  205.16
Permanent Ineff=
       F       F
Bank Sta=3821.8,6476.6
XS Rating Curve= 0 ,0
Exp/Cntr=0.3,0.1

Type RM Length L Ch R = 1 ,14000   ,500,500,500
BEGIN DESCRIPTION:
BELL CREEK 28.0
END DESCRIPTION:
XS GIS Cut Line= 3
      3807168.69     10137768.63      3805494.54     10138547.82
      3803282.33     10139095.95
#Sta/Elev= 30
  3153.4  232.37  3285.4  231.15    3397   228.4    3419  228.88  3576.4   220.1
  3719.2  209.18  3749.9  206.16  3856.5  201.27  3907.8  201.24  3908.8   199.9
  3921.9   199.9  3930.7     201  6239.1     201  6244.2  202.78  6263.8  205.95
  6280.5  211.06  6285.6  210.26  6346.2  211.42  6387.4  210.66  6409.8  212.92
  6489.5  212.87    6645  214.48  6818.6  219.83  6989.3  222.59  7113.5  226.77
  7149.8   229.2  7154.9  228.86  7170.4   230.9  7232.2  233.03  7279.1  232.46
#Mann= 4 ,-1 , 0
  3153.4     .11       0  3749.9     .06       0  6263.8    .125       0
  6489.5     .11       0
Bank Sta=3749.9,6263.8
XS Rating Curve= 0 ,0
Exp/Cntr=0.3,0.1

Type RM Length L Ch R = 1 ,13500   ,500,500,500
BEGIN DESCRIPTION:
BELL CREEK 27.0
END DESCRIPTION:
XS GIS Cut Line= 3
       3807105.1     10137697.08      3805264.43     10138103.92
      3803265.61     10139032.55
#Sta/Elev= 30
  3114.9  232.85  3173.5  232.79  3255.5  231.28  3337.1  226.15  3342.2  226.43
    3450  217.59  3483.4   216.1  3527.1  212.08  3668.2   203.4  3726.6  202.15
  3736.8  200.84  5003.4     201  6259.1  200.61  6259.6  200.11  6273.1  200.11
  6275.3  201.07  6297.4  203.38  6312.2  204.62  6335.1  208.78  6341.5  209.21
  6396.6  210.21  6506.9  214.48  6809.5  222.53  6878.2  225.46  6929.5  226.56
  6946.8  227.59    6981   227.8  7089.7  231.32  7102.3  232.26    7204  231.67
#Mann= 3 , 0 , 0
  3114.9     .11       0  3668.2     .06       0  6297.4     .11       0
Bank Sta=3668.2,6297.4
XS Rating Curve= 0 ,0
Exp/Cntr=0.3,0.1

Type RM Length L Ch R = 1 ,13000   ,500,500,500
BEGIN DESCRIPTION:
BELL CREEK 26.0
END DESCRIPTION:
XS GIS Cut Line= 3
      3807097.16     10137617.58      3805108.23     10137634.23
      3803251.27     10138951.96
#Sta/Elev= 30
    3011  233.25  3120.3  231.41  3180.3  226.32  3270.3  220.28  3420.3  208.74
  3470.3  206.64  3520.3  203.52  3540.3  203.15  3600.3  202.38  3620.3  200.97
  5004.9     201    6346  200.23  6346.5  199.73    6360  199.73  6361.5  201.85
    6368  203.21  6382.7  206.03  6388.9  205.98  6418.4  209.38  6590.7  215.67
  6819.5  221.53  6834.2  222.82  6869.9   224.2  6884.7  226.25  6913.3  227.15
  6920.3  228.14  7035.9  229.74  7092.6  228.84  7184.8  230.62    7277  229.89
#Mann= 3 , 0 , 0
    3011     .11       0  3540.3     .06       0    6368     .11       0
Bank Sta=3540.3,6368
XS Rating Curve= 0 ,0
Exp/Cntr=0.3,0.1

Type RM Length L Ch R = 1 ,12500   ,500,500,500
BEGIN DESCRIPTION:
BELL CREEK 25.0
END DESCRIPTION:
XS GIS Cut Line= 3
      3806954.05     10136647.77      3804981.39     10137151.27
      3803202.42     10138889.07
#Sta/Elev= 30
  2964.1  225.58    3043  225.99  3160.4  222.02  3237.9  221.43  3291.4     221
  3476.2  216.98  3528.1   209.8  3558.7     209  3569.1  210.53  3604.7  209.86
  3672.3  204.59  3703.3   200.8  6466.2  200.99  6473.6  199.77  6487.1  199.77
  6515.6  204.24  6536.9  207.41  6565.2  209.55  6664.2  213.66  6826.8   216.2
  6911.7  220.05  6918.8  219.24    6933  219.83  6982.4  223.82    7046  225.66
    7237  226.38  7272.3  227.45  7293.6  226.79    7442  229.22  7486.9  228.31
#Mann= 5 ,-1 , 0
  2964.1     .11       0  3237.9     .17       0  3291.4     .11       0
  3672.3     .06       0  6515.6     .11       0
Bank Sta=3672.3,6515.6
XS Rating Curve= 0 ,0
Exp/Cntr=0.3,0.1

Type RM Length L Ch R = 1 ,12000   ,500,500,500
BEGIN DESCRIPTION:
BELL CREEK 24.0
END DESCRIPTION:
XS GIS Cut Line= 3
       3806532.8     10134938.63      3804835.08     10136673.15
       3803117.9     10136611.07
#Sta/Elev= 30
  2572.9  230.13  2585.2  228.85  2592.2  225.61  2606.4  224.72  2648.8   226.4
  2781.8  222.44    2854  219.81  2868.1  218.03  2875.1  219.22  2882.3  216.69
  2889.2  217.13  2896.4  215.48  2972.5  214.07  2988.3  212.39  2995.4  208.03
  3016.5  206.46    3059  206.69  3073.1   203.2  3094.3  202.38  3108.7  200.06
  3129.7     201    6168     201    6188  203.33  6268.1   206.6  6388.1  207.07
  6478.2  211.28  6528.2   215.4  6598.3  216.48  6648.3  219.93  6718.3  221.44
#Mann= 5 ,-1 , 0
  2572.9     .15       0  2781.8    .125       0  2972.5     .11       0
  3073.1     .06       0    6188     .11       0
Bank Sta=3073.1,6188
XS Rating Curve= 0 ,0
Exp/Cntr=0.3,0.1

Type RM Length L Ch R = 1 ,11500   ,500,500,500
BEGIN DESCRIPTION:
BELL CREEK 23.0
END DESCRIPTION:
XS GIS Cut Line= 3
      3806477.12     10134898.92      3804688.72     10136195.05
      3803098.71     10136528.51
#Sta/Elev= 30
  2791.3  231.57  2900.6  230.31  2906.7  227.68  2921.4  229.67  2927.6  226.55
  2942.3  225.79  2950.8  226.65    2957  225.31  3042.8  222.29  3057.5   223.4
  3128.6  215.63  3164.2  214.24  3243.9   214.1  3258.6  212.08  3272.1  208.04
  3285.6  206.42  3344.4   204.9  3365.3  203.75  3371.4  201.26  3379.3   200.4
  6094.2     201  6145.2  204.77  6222.4  206.89  6317.1  207.18  6380.3  210.88
  6400.7  210.52  6416.9  213.49  6441.6   215.9  6516.7     217  6624.6  221.75
#Mann= 3 , 0 , 0
  2791.3    .125       0  3344.4     .06       0  6145.2     .11       0
Bank Sta=3344.4,6145.2
XS Rating Curve= 0 ,0
Exp/Cntr=0.3,0.1

Type RM Length L Ch R = 1 ,11000   ,500,500,500
BEGIN DESCRIPTION:
BELL CREEK 22.0
END DESCRIPTION:
XS GIS Cut Line= 3
      3806453.28     10134843.27      3804665.18     10135696.64
      3803074.78     10136449.05
#Sta/Elev= 30
  3018.7  232.31  3044.9  230.97  3135.5  230.81  3169.4  229.66  3192.1  227.95
  3214.8  224.87  3243.3  223.88  3278.3  223.86  3305.5  223.75  3328.2  221.57
  3368.1  219.52  3441.7  213.26    3538  214.33  3555.1  212.78  3589.8  207.52
    3612  208.02  3634.3  206.71  3674.1  206.25  3696.8  204.49  3718.2  200.49
  6211.5     201  6239.8  204.16  6285.3  206.26  6336.3  207.38  6413.1     207
  6490.1  210.62  6512.6  210.09  6518.4  211.41  6677.7  220.16  6759.4  223.02
#Mann= 5 ,-1 , 0
  3018.7    .125       0  3243.3     .11       0  3278.3    .125       0
  3696.8     .06       0  6239.8     .11       0
Bank Sta=3696.8,6239.8
XS Rating Curve= 0 ,0
Exp/Cntr=0.3,0.1

Type RM Length L Ch R = 1 ,10500   ,500,500,500
BEGIN DESCRIPTION:
BELL CREEK 21.0
END DESCRIPTION:
XS GIS Cut Line= 3
      3806413.58     10134795.56      3804535.18     10135225.62
      3803043.01     10136393.39
#Sta/Elev= 30
    3073  230.15  3232.8  229.18    3243   227.6  3251.3   224.8    3276  223.76
  3347.4  223.81  3390.4   222.3  3454.5  216.82  3540.5  215.03  3586.6  211.95
  3615.2   211.1  3701.1     205    3792  203.02  3800.4  200.49  6277.7     201
    6284  201.17  6291.8  203.28  6327.4  205.62  6383.5  205.76  6441.3  207.18
  6447.7  208.25  6497.4   207.2  6533.1  208.91  6540.8   210.2  6583.9  210.55
    6605  213.95  6625.8  213.25  6669.2   216.1  6832.9   223.2  6894.8  223.67
#Mann= 6 ,-1 , 0
    3073    .125       0    3276     .11       0  3454.5    .125       0
  3586.6     .11       0    3792     .06       0  6291.8     .11       0
Bank Sta=3792,6291.8
XS Rating Curve= 0 ,0
Exp/Cntr=0.3,0.1
