HEC-RAS study MCDONALD CREEK.prj: MCDONALD CREEK Base Level Engineering

--- MCDONALD CREEK.g01 (geometry) --- (continued)

Type RM Length L Ch R = 1 ,44500   ,500,500,500
BEGIN DESCRIPTION:
MCDONALD CREEK 87.0
END DESCRIPTION:
XS GIS Cut Line= 3
      3792823.82     10232093.07        3792288.      10232886.6
      3791914.08     10233454.21
#Sta/Elev= 30
  4042.5  357.79  4088.4  354.55  4132.1  349.87  4138.1  350.51    4255   342.9
  4290.9  338.56  4332.9   337.2  4347.9  335.19  4353.9  336.22  4362.9  334.77
  4422.2  333.14  4485.7  327.71  4519.6  326.59  4609.3  322.61  4650.6  319.06
  4686.6  316.65  5005.8  315.48  5082.6  316.68  5112.8  319.01  5154.9  323.04
    5170  326.56  5211.5  328.79  5227.2  328.32  5233.2  330.65  5248.3  333.01
  5364.6   341.2  5400.5  342.68  5508.3  352.49  5594.6  356.64  5679.7  357.82
#Mann= 7 ,-1 , 0
  4042.5     .17       0  4422.2     .11       0  4519.6     .17       0
  4609.3     .11       0  4650.6    .015       0  5112.8     .11       0
  5211.5     .11       0
Bank Sta=4650.6,5112.8
XS Rating Curve= 0 ,0
Exp/Cntr=0.3,0.1

Type RM Length L Ch R = 1 ,44000   ,500,500,500
BEGIN DESCRIPTION:
MCDONALD CREEK 86.0
END DESCRIPTION:
XS GIS Cut Line= 3
      3792452.11     10231946.27      3791934.44     10232533.05
      3791868.75     10233232.78
#Sta/Elev= 30
  4217.5  348.85    4306  343.76  4365.7  337.61  4400.9  334.95  4415.1   332.7
  4443.5  330.74  4464.4  327.13  4478.6  325.67    4564  319.54  4570.7  318.48
  4578.2  318.63  4606.7  315.84  4861.8  315.68    4864  315.16  4917.9     316
  5078.4  315.73  5118.5  316.42  5188.8   319.3  5259.2  323.85  5299.3  325.16
  5309.4  324.87  5341.2  326.82  5389.7  328.38  5419.9  330.66    5445  330.97
  5500.2  334.31  5540.4  337.61  5560.5  341.15  5630.8  342.42  5702.8  349.08
#Mann= 4 ,-1 , 0
  4217.5     .17       0    4306     .11       0    4564    .015       0
  5188.8     .11       0
Bank Sta=4564,5188.8
XS Rating Curve= 0 ,0
Exp/Cntr=0.3,0.1

Type RM Length L Ch R = 1 ,43500   ,500,500,500
BEGIN DESCRIPTION:
MCDONALD CREEK 85.0
END DESCRIPTION:
XS GIS Cut Line= 3
      3792155.19     10231821.31      3791633.38     10232136.27
      3791118.78     10232165.05
#Sta/Elev= 30
  4390.5  342.88  4402.3  339.84  4408.5   339.7  4433.3  340.56  4454.7  339.75
  4488.5  335.53  4504.2  333.44  4534.3  331.97  4555.6  328.93    4586  326.89
  4598.4  324.18    4608   323.5  4629.4   320.6  4635.2  319.42  4656.6  317.26
  4899.2  316.92  5035.6  315.61  5180.8  315.43  5181.3  314.93  5190.4  314.93
  5195.8  315.72  5225.9  315.92    5276  319.93    5296  323.43  5336.1  325.11
  5352.9   328.4  5395.2   333.1  5456.2  337.76  5486.3  338.44  5515.4  337.32
#Mann= 6 ,-1 , 0
  4390.5     .11       0  4408.5     .17       0  4488.5     .11       0
  4629.4    .015       0    5276     .11       0  5395.2     .11       0
Bank Sta=4629.4,5276
XS Rating Curve= 0 ,0
Exp/Cntr=0.3,0.1

Type RM Length L Ch R = 1 ,43000   ,500,500,500
BEGIN DESCRIPTION:
MCDONALD CREEK 84.0
END DESCRIPTION:
XS GIS Cut Line= 3
      3792139.58     10231753.59       3791340.4     10231731.11
      3791087.52     10232066.07
#Sta/Elev= 30
  4200.5  342.07  4222.2  340.56  4252.2  340.43  4292.3  338.39  4342.3  332.65
  4372.3  330.18  4412.3  327.62  4432.3  327.45  4467.6  324.14  4482.3  324.17
  4507.5  321.95  4532.4  319.96  4562.4  319.07  4592.4  317.66  4662.4  315.96
  4752.4  316.22    4847  315.49  4847.5  314.99  4972.5  316.38  5144.7  315.87
  5159.2  316.28  5187.9  319.17  5223.8  322.98    5230  324.51  5259.1  327.13
  5265.4  328.38  5273.7  328.55  5315.4   333.5  5388.2  338.07  5419.7  337.58
#Mann= 4 ,-1 , 0
  4200.5     .17       0  4507.5     .11       0  4562.4    .015       0
  5187.9     .11       0
Bank Sta=4562.4,5187.9
XS Rating Curve= 0 ,0
Exp/Cntr=0.3,0.1

Type RM Length L Ch R = 1 ,42500   ,629,629,629
BEGIN DESCRIPTION:
MCDONALD CREEK 83.0
END DESCRIPTION:
XS GIS Cut Line= 4
      3791972.93     10230894.21      3791145.41     10231286.02
      3791121.86      10231337.1      3791040.84     10232027.82
#Sta/Elev= 30
  4084.4  337.55  4092.2  336.09  4160.4  333.48  4245.3   331.2  4325.2  328.65
  4342.4  328.76  4365.1  327.41  4412.2  326.22  4461.3  324.79  4521.5  324.05
  4529.9  323.28  4535.4  321.21  4575.4  319.38  4587.9  317.93  4598.2  317.91
  4603.7  317.05  4626.4  315.92    4776  316.98  4876.7  315.85  4877.2  315.35
  4904.9  316.27  5332.1  316.42  5362.3   318.3  5394.3  319.35  5452.9  323.63
  5493.2  328.26  5603.9  333.77  5684.5  335.98  5724.8  336.23  5751.7  335.09
#Mann= 6 ,-1 , 0
  4084.4     .17       0  4245.3     .11       0  4412.2     .17       0
  4461.3     .11       0  4575.4    .015       0  5394.3     .11       0
Bank Sta=4575.4,5394.3
XS Rating Curve= 0 ,0
Exp/Cntr=0.3,0.1

Type RM Length L Ch R = 1 ,41871   ,371,371,371
XS GIS Cut Line= 4
      3791150.19      10230252.7      3790961.92      10230710.8
      3790697.29     10231459.94      3791000.21     10232000.52
#Sta/Elev= 30
       0  346.16    22.3  345.37    70.2  346.49   160.4  344.87   206.3  342.96
   236.1  339.88   246.9  339.73   259.6   341.7   283.6  341.14   376.6  332.95
   398.3  325.02   413.9  321.13   419.9  318.04   443.6  315.26   473.9  314.33
   506.2  315.06     538  318.95     591  320.58   702.5  321.11  1093.9  320.58
  1181.3  321.45  1243.2  320.31  1336.6  321.83  1401.7  321.21  1542.1  324.29
  1577.7   326.2  1600.6   325.8  1644.8  328.74  1715.6  331.11  1909.5  335.03
#Mann= 3 , 0 , 0
       0     .11       0   419.9     .07       0     538     .11       0
Bank Sta=419.9,538
XS Rating Curve= 0 ,0
Exp/Cntr=0.3,0.1

Type RM Length L Ch R = 1 ,41500   ,500,500,500
BEGIN DESCRIPTION:
MCDONALD CREEK 81.0
END DESCRIPTION:
XS GIS Cut Line= 3
      3791071.86     10230222.35      3790737.98     10230425.83
      3790014.59     10232185.87
#Sta/Elev= 30
    4609  342.39  4675.1   339.2  4687.7  338.24    4887  327.25  4945.1  321.66
  4953.3  318.33  4988.4  313.96  5027.3  313.57  5059.7  314.79  5081.4  318.61
    5103  318.94  5118.9  312.89  5135.4  310.89  5302.1  302.42  5373.3  299.93
  5481.4   299.1    5503  300.87  5516.3  298.27  5519.5  292.68  5529.8  292.68
  5534.8  296.54  5546.3  300.51    5643  301.74  5831.6  304.23  5961.5  304.07
    6284  309.08  6513.4  318.66  6735.5  331.68  6791.4     337  6902.9  342.28
#Mann= 12 ,-1 , 0
    4609     .11       0  4675.1     .17       0  4687.7     .11       0
  4953.3     .07       0  5081.4     .11       0  5302.1     .15       0
    5503     .15       0  5546.3     .11       0    5643     .15       0
  5831.6     .11       0    6284     .17       0  6791.4     .11       0
Bank Sta=5503,5546.3
XS Rating Curve= 0 ,0
Exp/Cntr=0.3,0.1

Type RM Length L Ch R = 1 ,41000   ,505,505,505
BEGIN DESCRIPTION:
MCDONALD CREEK 80.0
END DESCRIPTION:
XS GIS Cut Line= 3
       3790686.5     10229873.35      3790341.93     10230168.82
      3789946.88      10232154.6
#Sta/Elev= 30
  4546.1  341.23  4636.2  336.91    4870  318.11  4898.5   314.6  4968.8  311.42
  5003.7  312.71  5032.9  317.95  5047.4  317.87  5083.9  309.65  5114.5   305.8
  5338.8  298.68  5399.9  296.57  5405.1  292.06  5415.4  292.06  5420.3     296
  5430.5  299.27  5499.6  298.67    5763  301.08  5921.4  313.83  5981.1  315.24
    6177  303.81  6330.4  304.61  6483.8  311.63  6552.1  314.28  6580.8  317.43
  6643.9  317.87  6683.1  322.15  6863.6  332.27  6949.7  339.69  7024.7  342.99
#Mann= 8 ,-1 , 0
  4546.1     .11       0    4870     .07       0  5032.9     .11       0
  5338.8     .15       0  5430.5     .15       0  5499.6     .11       0
  6483.8     .17       0  6863.6     .11       0
Bank Sta=5338.8,5430.5
XS Rating Curve= 0 ,0
Exp/Cntr=0.3,0.1

Type RM Length L Ch R = 1 ,40495   ,451,451,451
BEGIN DESCRIPTION:
MCDONALD CREEK 77.0
END DESCRIPTION:
XS GIS Cut Line= 3
      3790071.87     10229842.13      3789847.12     10230101.51
      3788717.84     10231661.08
#Sta/Elev= 30
  4656.8  332.04  4807.8  325.26  4899.9   318.1  4928.4  317.94  4971.2  313.57
  5006.5  307.33  5071.4   307.3  5098.5  303.71  5145.9  300.49  5196.5  297.69
  5257.8  296.95  5293.4  294.32  5293.9  291.91  5294.4  291.41  5304.7  291.41
  5314.2  295.63  5320.5  296.55  5370.7  296.68  5406.2  295.24  5483.5  295.12
  5593.4  294.01  5693.2  293.89  5758.1  295.82  5851.4  295.31  5944.5  299.84
  6130.9  305.91  6545.4  313.87  6574.8  316.33  6802.9  322.65  6925.5  327.68
#Mann= 8 ,-1 , 0
  4656.8     .11       0  5145.9     .17       0  5196.5     .11       0
  5257.8     .06       0  5320.5     .11       0  5406.2     .11       0
  5483.5     .15       0  5593.4     .11       0
Bank Sta=5257.8,5320.5
XS Rating Curve= 0 ,0
Exp/Cntr=0.3,0.1

Type RM Length L Ch R = 1 ,40044   ,948,948,948
BEGIN DESCRIPTION:
MCDONALD CREEK 76.0
END DESCRIPTION:
XS GIS Cut Line= 3
      3789767.87     10229761.06      3789409.69     10229996.61
      3788524.98     10231284.88
#Sta/Elev= 30
  4571.3  319.62  4795.8  302.98  4955.6  295.55  4961.5  295.53  5017.8  293.88
  5083.5   295.5  5090.3  294.92  5099.3  291.02  5109.6  291.02  5134.3  295.34
  5349.4  291.68  5695.9  294.68  5860.3  300.04  5946.9  299.94  5997.7  301.85
  6018.7  300.31  6024.7  301.81  6060.8  300.98  6075.5  302.49  6084.3  301.02
  6105.3  303.31  6120.2   301.9  6147.2  305.88    6170  303.72    6177  306.39
  6191.9  307.59  6206.4  306.33  6212.9  308.32  6341.4  313.59  6562.8  317.56
#Mann= 4 ,-1 , 0
  4571.3     .11       0  4955.6     .17       0  4961.5     .07       0
  5134.3     .12       0
#XS Ineff= 2 , 0
       0                  5722.9       0  296.45
Permanent Ineff=
       F       F
Bank Sta=4961.5,5134.3
XS Rating Curve= 0 ,0
Exp/Cntr=0.3,0.1

Type RM Length L Ch R = 1 ,39096   ,479,479,479
BEGIN DESCRIPTION:
MCDONALD CREEK 75.0
END DESCRIPTION:
XS GIS Cut Line= 3
      3789660.42     10229675.46      3788766.92     10229527.93
      3788051.92     10230179.87
#Sta/Elev= 30
  4094.4   314.1  4147.3  308.83    4249  302.34  4350.4  300.09  4370.7  298.41
  4411.2  298.35  4441.6  295.93    4524  294.37  4573.4  296.04  4634.2  292.82
  4674.7  289.07  4695.8  290.32  4763.4  289.35  4796.3  290.85  4816.6  289.17
  4890.6  289.17    4902  288.09  4978.8  290.25  5015.6  289.31    5023  291.12
  5100.7  289.75    5150  291.72    5200  291.24  5249.3  293.89  5334.5  294.37
  5518.2  301.97  5560.8  305.23  5681.1  308.12  5837.1  314.81  5967.6  318.41
#Mann= 4 ,-1 , 0
  4094.4     .11       0  4695.8     .17       0  4796.3     .06       0
    5023     .11       0
Bank Sta=4796.3,5023
XS Rating Curve= 0 ,0
Exp/Cntr=0.3,0.1

Type RM Length L Ch R = 1 ,38617   ,478,478,478
BEGIN DESCRIPTION:
MCDONALD CREEK 74.0
END DESCRIPTION:
XS GIS Cut Line= 3
      3789764.62     10229269.22      3788925.38     10229092.72
      3787801.93     10229799.91
#Sta/Elev= 30
  4142.4  314.93  4161.2  310.79  4190.2  312.18  4231.1  310.59  4300.5  305.03
  4343.5  304.55  4394.6   301.8  4444.9  298.36  4455.9  296.24  4486.5  295.68
  4544.6  291.79  4782.9  285.99  4813.5  287.16  4827.1  285.65  4827.6  285.15
  4839.8  285.65    4988   287.7  4996.2  285.84  5010.5  285.71  5032.5  287.76
  5171.8  286.82  5229.5  288.77  5235.4  290.27  5271.9  292.14  5351.6  293.34
  5375.2  294.99  5721.7  300.59  5867.7  305.28  6034.9  307.47  6327.5  315.43
#Mann= 5 ,-1 , 0
  4142.4     .11       0  4827.1     .09       0  4839.8     .11       0
    4988     .06       0  5032.5     .11       0
Bank Sta=4988,5032.5
XS Rating Curve= 0 ,0
Exp/Cntr=0.3,0.1

Type RM Length L Ch R = 1 ,38139   ,498,498,498
BEGIN DESCRIPTION:
MCDONALD CREEK 73.0
END DESCRIPTION:
XS GIS Cut Line= 3
       3790167.9     10228561.07      3788972.14      10228669.9
      3787623.96     10229519.21
#Sta/Elev= 30
  3799.3  351.98  3854.5  348.82  3959.9  338.71  3964.9  339.26  4020.3  335.14
  4060.4  329.58  4075.3  328.53  4100.6  323.81  4180.7  316.64  4185.7  317.67
    4211  313.42  4291.1  310.28  4331.5  305.58  4361.7  305.16  4532.4  292.26
  4662.9  288.24  4763.3  286.51  4903.9  285.06  4984.2  286.03  4988.4  283.42
  5000.2  283.42  5005.5  285.89    5206  284.91  5236.1  286.47  5293.8  284.95
  5570.4  293.35  5764.7  296.41  5874.2  299.93  6004.8  305.76  6593.4  314.06
#Mann= 3 , 0 , 0
  3799.3     .11       0  4984.2     .07       0  5005.5     .11       0
#XS Ineff= 2 , 0
       0  4672.9  288.42               0
Permanent Ineff=
       F       F
Bank Sta=4984.2,5005.5
XS Rating Curve= 0 ,0
Exp/Cntr=0.3,0.1

Type RM Length L Ch R = 1 ,37641   ,499,499,499
BEGIN DESCRIPTION:
MCDONALD CREEK 72.0
END DESCRIPTION:
XS GIS Cut Line= 3
      3789367.88     10227611.04      3788769.34     10228224.39
      3787655.24     10229316.06
#Sta/Elev= 30
    4143  312.61  4178.4  309.03  4206.7  307.91    4242  304.66  4277.4  303.38
  4284.4  302.17  4326.8  298.83  4418.9  294.31  4524.9  291.57  4574.5  288.57
  4694.6  286.36  4991.7  284.16  4999.7  281.86  5011.7  281.86  5012.2  282.36
  5012.9  284.66    5123  284.06  5486.7   282.5    5621  286.16    5720  289.82
  5741.2  291.29  5748.2  290.75    5784  292.82    5809  294.18  5894.4  297.59
  5960.4  301.36  6031.1  302.55  6108.9  305.78  6196.5  307.51  6559.8  311.42
#Mann= 8 ,-1 , 0
    4143     .11       0  4991.7     .06       0  5012.9     .11       0
    5123     .15       0    5784     .17       0    5809     .15       0
  5894.4     .17       0  6196.5     .11       0
Bank Sta=4991.7,5012.9
XS Rating Curve= 0 ,0
Exp/Cntr=0.3,0.1

Type RM Length L Ch R = 1 ,37142   ,499,499,499
BEGIN DESCRIPTION:
MCDONALD CREEK 71.0
END DESCRIPTION:
XS GIS Cut Line= 3
      3789109.23     10227333.32      3788549.01     10227791.62
      3787367.87     10228511.06
#Sta/Elev= 30
  4276.2  306.89  4510.5   297.7  4624.2  295.32    4645  293.44  4822.3  284.76
  4943.6  282.53  4986.7  283.02  4993.1  282.63  4997.5  280.86  5003.6  280.86
  5013.7  283.13    5066  281.52  5118.2  282.03  5160.9  280.69  5277.1  279.86
  5319.7   281.7  5364.3  280.88    5381  279.21  5381.5  278.71    5394  279.21
  5399.5  280.78  5412.4  280.62  5466.9  280.39  5619.9  282.81  5647.1  284.73
  5720.6  286.13  5794.2  289.72  6072.2  299.02  6164.2  302.99    6383  308.28
#Mann= 7 ,-1 , 0
  4276.2     .11       0  4986.7     .06       0  5013.7     .15       0
    5381     .09       0    5394     .15       0  5412.4     .17       0
  6072.2     .11       0
#XS Ineff= 2 , 0
       0                  5699.3       0  286.06
Permanent Ineff=
       F       F
Bank Sta=4986.7,5013.7
XS Rating Curve= 0 ,0
Exp/Cntr=0.3,0.1

Type RM Length L Ch R = 1 ,36643   ,475,475,475
BEGIN DESCRIPTION:
MCDONALD CREEK 70.0
END DESCRIPTION:
XS GIS Cut Line= 3
      3788973.79     10227109.38      3788333.94     10227363.05
      3787217.86     10228261.06
#Sta/Elev= 30
  4311.7  308.38  4640.8  302.11    4956  281.86  4985.7  280.53  5009.5  281.72
  5110.3  280.04  5159.9  281.61  5195.1  279.66  5273.3  278.82  5407.1  278.69
  5409.3  278.59  5409.8  278.09  5422.3  278.59  5614.2  281.34  5678.2  284.45
  5735.8  285.16  5884.6  293.08  5934.2  294.07  5948.6  295.71    5963   295.1
  6139.3   301.3  6175.8  302.16  6183.7  299.87  6198.1  299.29  6226.9  300.73
  6270.1   300.5  6297.3  301.56  6311.7  305.18  6318.1  304.46  6432.5  308.42
#Mann= 9 ,-1 , 0
  4311.7     .11       0    4956     .07       0  5159.9     .15       0
  5273.3     .15       0  5407.1     .17       0  5409.3     .09       0
  5422.3     .17       0  6139.3     .11       0  6270.1     .17       0
Bank Sta=4956,5159.9
XS Rating Curve= 0 ,0
Exp/Cntr=0.3,0.1

Type RM Length L Ch R = 1 ,36168   ,491,491,491
BEGIN DESCRIPTION:
MCDONALD CREEK 69.0
END DESCRIPTION:
XS GIS Cut Line= 3
      3788895.63     10226791.68      3788088.44     10226983.64
       3786973.8     10227776.04
#Sta/Elev= 30
  4170.3  306.97  4275.8  303.87  4435.3  294.98    4610  290.12  4774.5  283.46
  4889.6  280.12  4971.1  280.38  4997.7  278.65  5020.3     280  5098.9  277.96
  5154.4  278.23    5165  277.89  5165.5  277.39  5178.1  277.89  5299.5  279.09
  5456.9  284.04  5601.9  285.08  5643.8  287.01    5651  287.07  5658.6  285.36
  5679.5  286.45  5694.2  285.36  5723.8  288.07  5757.1  288.78    5816  289.02
  5849.9  290.42  6068.1   292.1  6225.6   296.3  6353.4  302.74  6367.6  302.48
#Mann= 9 ,-1 , 0
  4170.3     .11       0  4889.6     .15       0  4971.1     .09       0
  5020.3     .15       0  5154.4     .11       0    5165     .12       0
  5178.1     .11       0  5757.1     .15       0  5849.9     .11       0
Bank Sta=4971.1,5020.3
XS Rating Curve= 0 ,0
Exp/Cntr=0.3,0.1

Type RM Length L Ch R = 1 ,35677   ,494,494,494
BEGIN DESCRIPTION:
MCDONALD CREEK 68.0
END DESCRIPTION:
XS GIS Cut Line= 3
      3788467.82      10226161.1      3787851.05     10226722.19
      3786859.21     10227218.76
#Sta/Elev= 30
  4166.2  312.58    4230  309.06  4272.6  305.23  4293.5   301.9  4378.7  295.87
  4435.4  290.04  4442.2  287.53  4449.6  286.51  4456.4  288.22  4484.7  287.87
  4491.5  285.83  4531.7  281.84  4558.7  280.82  4647.6  278.49  4733.9  278.46
  4930.7  278.42  4973.3  277.84  4981.3  276.46  4998.8   277.6  5104.2  278.38
  5254.8  279.32  5283.2  281.25  5344.2  281.28  5388.9   284.1  5450.4  284.08
  5612.4  291.03    5641  293.46  5763.3  296.64  5986.8  305.23  6109.2  307.96
#Mann= 6 ,-1 , 0
  4166.2     .11       0  4531.7     .15       0  4558.7     .11       0
  4733.9     .15       0  4930.7     .09       0  5104.2     .15       0
Bank Sta=4930.7,5104.2
XS Rating Curve= 0 ,0
Exp/Cntr=0.3,0.1

Type RM Length L Ch R = 1 ,35183   ,498,498,498
BEGIN DESCRIPTION:
MCDONALD CREEK 67.0
END DESCRIPTION:
XS GIS Cut Line= 3
      3788421.69     10226098.97      3787908.19     10226271.78
      3786817.55     10227041.67
#Sta/Elev= 30
  4458.2  313.11  4504.5  311.48  4567.8  306.75  4579.1  304.58  4599.4  303.81
  4699.8  293.09  4752.6  289.43  4799.9  285.43  4825.8   287.3  4863.2  280.54
  4894.8  277.37  4946.5  276.75  4968.7  277.74    4978  277.22  4983.6  274.05
  4996.1  274.05  4997.5  276.02    5007  276.94  5013.1  275.83  5021.8  276.94
  5099.3  277.44  5200.3  275.83  5235.4  277.02  5245.7  276.43  5696.5  286.13
  5788.8  288.74  5904.6  293.95  6032.6  297.15  6163.2  302.73    6335  307.07
#Mann= 6 ,-1 , 0
  4458.2     .11       0  4752.6     .15       0  4968.7     .06       0
  5099.3     .15       0  5235.4     .15       0  5245.7     .11       0
Bank Sta=4968.7,5099.3
XS Rating Curve= 0 ,0
Exp/Cntr=0.3,0.1

Type RM Length L Ch R = 1 ,34685   ,498,498,498
BEGIN DESCRIPTION:
MCDONALD CREEK 66.0
END DESCRIPTION:
XS GIS Cut Line= 3
      3788385.29     10225875.01      3787786.17     10225809.42
      3786366.12      10226306.7
#Sta/Elev= 30
  4397.3  310.72    4445  307.27  4465.1  304.72  4495.3  303.27  4585.9  294.17
  4656.3  290.05  4696.5   286.7  4706.6  284.84    4759  281.84  4887.6  274.88
  4958.1  275.44  4988.2  273.16    5000  273.58  5008.8  275.28  5115.5   274.6
  5135.9  273.53  5203.3  274.51  5241.9   273.9  5246.3  272.02  5259.3  272.52
    5260  273.51  5446.1  276.53  5539.2  282.28    5627  284.43  5683.7  284.08
  5792.9  289.16  6057.8  297.84  6226.2  301.86  6355.6  302.75  6504.6  309.83
#Mann= 5 ,-1 , 0
  4397.3     .17       0    4759     .11       0  4958.1     .06       0
  5008.8     .15       0  5259.3     .11       0
Bank Sta=4958.1,5008.8
XS Rating Curve= 0 ,0
Exp/Cntr=0.3,0.1

Type RM Length L Ch R = 1 ,34187   ,439,439,439
BEGIN DESCRIPTION:
MCDONALD CREEK 65.0
END DESCRIPTION:
XS GIS Cut Line= 3
       3788317.5     10225203.14      3787610.74     10225401.62
      3786364.42     10226203.13
#Sta/Elev= 30
  4265.9  301.05  4369.4  297.37  4431.7  293.99  4442.1  294.68  4464.9  292.88
  4566.8  289.68  4577.5     288  4679.7  283.04  4754.1  278.34  4857.7  274.34
  4888.7  273.16  4971.8  273.11  4992.6  268.93  5005.2  268.93  5008.8  270.37
  5015.3   270.9    5024  273.78  5033.7  273.32  5045.1  272.52  5051.1  273.18
  5348.2  272.74  5544.4  275.21    5617  280.76  5659.3  283.18  5674.5  283.11
  5704.9  285.98  5840.9  289.67  5949.9  294.73  6194.9   302.5  6481.8   309.7
#Mann= 6 ,-1 , 0
  4265.9     .17       0  4754.1     .11       0  4857.7     .15       0
  4971.8     .09       0    5024     .15       0  5033.7     .11       0
Bank Sta=4971.8,5024
XS Rating Curve= 0 ,0
Exp/Cntr=0.3,0.1

Type RM Length L Ch R = 1 ,33748   ,1046,1046,1046
BEGIN DESCRIPTION:
MCDONALD CREEK 64.0
END DESCRIPTION:
XS GIS Cut Line= 4
      3788317.49     10225130.22       3787397.9     10225120.73
      3787357.66      10225130.3      3786322.78     10226130.18
#Sta/Elev= 30
    4039  300.47  4318.7  294.81  4554.6  283.21  4598.7   282.9  4638.7  279.94
  4668.7  280.66  4890.9  272.38  4938.7  269.82    4969  272.05  4976.7  268.63
  4989.3  268.63  4997.3   271.2  5021.6  269.42  5028.6  272.07    5071  272.02
  5078.2  270.25    5084  271.63  5092.4  270.21  5113.5  272.05  5163.1  271.85
  5177.3  269.32  5205.6  271.56  5347.1  271.35  5502.4  274.31  5693.6  282.89
  5757.1  287.79  6004.6  297.41  6245.1  303.65  6308.7  302.23    6439  310.34
#Mann= 6 ,-1 , 0
    4039     .17       0  4554.6     .11       0  4890.9     .15       0
    4969     .09       0  5028.6     .15       0    5084     .11       0
Bank Sta=4969,5028.6
XS Rating Curve= 0 ,0
Exp/Cntr=0.3,0.1

Type RM Length L Ch R = 1 ,32702   ,497,497,497
BEGIN DESCRIPTION:
MCDONALD CREEK 63.0
END DESCRIPTION:
XS GIS Cut Line= 3
      3786950.56     10223541.17      3786580.67     10224975.75
      3786182.79     10225896.02
#Sta/Elev= 30
  3518.5  296.33    3570  292.51  3592.6  293.16  3606.2  291.54  3807.6  282.63
    3984  278.78  4220.6     273  4585.1  271.97  4716.3  271.18  4746.6   272.2
  4757.6  271.04  4819.6  272.16  4933.2   270.5  4955.1  268.86  4966.1  270.11
  4974.5  270.07  4984.8  269.13  4988.6  265.68  5002.6  265.68  5020.9  268.94
  5044.4  269.99  5180.1  271.85  5441.6  278.52    5594   283.7  5798.3  294.41
  5803.7  293.26  5874.2  297.17  5955.6  298.24  5986.3  301.39  6002.6  301.68
#Mann= 7 ,-1 , 0
  3518.5     .11       0  3606.2     .17       0    3984     .11       0
  4585.1     .15       0  4966.1     .11       0  4974.5     .06       0
  5044.4     .11       0
Bank Sta=4974.5,5044.4
XS Rating Curve= 0 ,0
Exp/Cntr=0.3,0.1

Type RM Length L Ch R = 1 ,32205   ,500,500,500
BEGIN DESCRIPTION:
MCDONALD CREEK 62.0
END DESCRIPTION:
XS GIS Cut Line= 3
      3786892.85     10223527.84      3786296.63     10224649.41
      3785481.94     10224832.89
#Sta/Elev= 30
  3729.8  296.94  3837.4  293.06    3877  287.53  3942.9  288.44  3959.2  286.99
  3964.9  287.87  4185.1   278.7  4231.8  275.68  4305.2  273.27  4541.3  270.02
    4569  270.66  4764.1  267.83  4859.6  270.32  4875.9  269.46  4979.2  270.88
  4985.8  270.63  4991.5  265.33  5001.9   264.1  5016.1   264.1  5019.2  268.72
  5039.8  271.35    5173  272.59  5294.4  278.24  5408.8  282.11  5442.3   282.1
  5572.1  290.53  5614.8   291.4  5716.9  296.54  5814.9  299.81  5835.1  300.33
#Mann= 10 ,-1 , 0
  3729.8     .11       0  3837.4     .17       0  4185.1     .11       0
    4569     .15       0  4979.2     .09       0  5039.8     .15       0
  5294.4     .17       0  5614.8     .11       0  5716.9     .17       0
  5814.9     .11       0
Bank Sta=4979.2,5039.8
XS Rating Curve= 0 ,0
Exp/Cntr=0.3,0.1

Type RM Length L Ch R = 1 ,31705   ,785,785,785
BEGIN DESCRIPTION:
MCDONALD CREEK 61.0
END DESCRIPTION:
XS GIS Cut Line= 3
      3786821.82     10223487.89      3786126.49     10224263.82
      3785411.46     10224707.89
#Sta/Elev= 30
  3958.1  297.85  3989.9  296.84  4096.4  292.06  4147.5  290.86  4196.8  286.83
  4345.6  282.69  4405.1  279.16  4451.8  275.17  4514.9  272.53  4543.7  270.76
    4770  268.76  4826.5  268.38  4869.7  267.69  4961.6  270.14  4975.8  269.42
  4982.9  260.79  4997.2  260.79  5010.2  265.48  5019.6  265.86  5040.9  269.89
  5046.8  271.17  5186.7  276.84  5403.4  288.88  5461.3  291.48  5497.9  292.07
  5504.6  291.01  5534.5  294.25  5613.1  296.88  5760.1  301.72  5841.7  302.38
#Mann= 10 ,-1 , 0
  3958.1     .11       0  3989.9     .17       0  4096.4     .11       0
  4405.1     .17       0  4514.9     .11       0    4770     .17       0
  4826.5     .15       0  4961.6     .09       0  5040.9     .17       0
  5613.1     .11       0
Bank Sta=4961.6,5040.9
XS Rating Curve= 0 ,0
Exp/Cntr=0.3,0.1

Type RM Length L Ch R = 1 ,30920   ,710,710,710
BEGIN DESCRIPTION:
MCDONALD CREEK 60.0
END DESCRIPTION:
XS GIS Cut Line= 3
       3786684.2      10223310.3      3785937.86     10223744.19
      3785344.05     10224556.98
#Sta/Elev= 30
  4136.7  298.02  4331.1  287.16  4411.4  285.24  4491.6  280.16  4523.1  280.26
  4770.8  270.06    4807  267.82    4903  267.46  4908.8  266.67  4918.7  262.77
  4930.6  266.69  4953.7  267.66  4976.9  265.99  4983.3  262.51    4989  263.56
  4998.2     259  5012.6     259  5020.1  261.79  5026.3   265.8  5033.3  267.56
  5091.3  267.49  5141.3  267.41  5277.3     273  5312.8  275.69  5377.6   277.2
    5641  291.85  5736.8  295.68  5800.1  298.18  5856.5  298.37  6006.6  301.98
#Mann= 6 ,-1 , 0
  4136.7     .17       0  4770.8     .15       0  4953.7     .09       0
  5033.3     .15       0  5091.3     .17       0  5736.8     .11       0
Bank Sta=4953.7,5033.3
XS Rating Curve= 0 ,0
Exp/Cntr=0.3,0.1

Type RM Length L Ch R = 1 ,30210   ,499,499,499
BEGIN DESCRIPTION:
MCDONALD CREEK 58.0
END DESCRIPTION:
XS GIS Cut Line= 3
       3786537.7       10223075.      3785668.42     10223314.63
       3785263.5     10224411.37
#Sta/Elev= 30
  4098.3   300.1  4274.5  291.38  4305.6  286.52  4347.1   287.4  4658.3  270.42
  4704.2   269.2  4807.7  265.01  4818.2  266.57  4834.6   263.8    4845  264.04
  4917.6  267.78  4938.4  265.21  4979.8  266.77  4990.5  258.17  5014.1  258.85
  5019.5  261.28  5044.6   263.1  5049.9  265.79  5092.6  265.38  5221.8  267.96
    5316  275.25    5348  275.58  5388.4  278.86  5449.2  280.89  5465.2  283.09
    5682   288.1  5742.8  291.92  5767.9  290.89  6088.4  298.92  6169.1  300.36
#Mann= 7 ,-1 , 0
  4098.3     .17       0  4704.2     .11       0  4807.7     .15       0
  4979.8     .09       0  5049.9     .15       0  5092.6     .17       0
  6088.4     .11       0
Bank Sta=4979.8,5049.9
XS Rating Curve= 0 ,0
Exp/Cntr=0.3,0.1

Type RM Length L Ch R = 1 ,29711   ,500,500,500
BEGIN DESCRIPTION:
MCDONALD CREEK 57.0
END DESCRIPTION:
XS GIS Cut Line= 3
      3786517.82     10222961.07      3785309.39     10223078.22
      3785156.97     10224331.38
#Sta/Elev= 30
  3785.9  299.37  3839.4  297.92  3876.3  294.39    4238  274.92  4344.2  270.45
  4479.1  266.78  4742.5  263.95  4830.7  263.43  4901.1  265.11  4941.6  263.96
  4982.1  265.57  4991.1  259.56    5023  260.37  5033.1  263.21  5051.2  265.17
  5132.9  266.33  5264.8  273.16    5436  276.37  5469.8  277.55  5486.4   279.6
  5638.2  284.05    5698  287.24    5839     290  5869.2  292.75  5889.4  291.87
  5939.7  294.17  5970.1  293.28  6070.7  296.98  6206.6  299.54  6262.4  300.52
#Mann= 7 ,-1 , 0
  3785.9     .17       0  4344.2     .15       0  4742.5     .11       0
  4941.6     .17       0  4982.1     .09       0  5051.2     .17       0
  6206.6     .11       0
Bank Sta=4982.1,5051.2
XS Rating Curve= 0 ,0
Exp/Cntr=0.3,0.1

Type RM Length L Ch R = 1 ,29211   ,498,498,498
BEGIN DESCRIPTION:
MCDONALD CREEK 56.0
END DESCRIPTION:
XS GIS Cut Line= 3
       3785898.4     10221973.96      3785158.08     10222717.57
      3784221.57     10223500.07
#Sta/Elev= 30
  3950.7  297.59  4183.6  283.53  4201.8  282.45  4281.4  278.25  4359.2  270.75
  4415.7  268.59  4806.6  262.88  4882.4  260.76  4962.2  263.48  4974.4     264
  4988.5  262.39  4995.6  258.06  5002.6  256.46  5017.5  256.46  5024.4  265.18
  5045.2  264.36  5073.8  268.74  5102.4  269.99  5232.6  266.81  5250.8  266.76
  5272.9  263.32  5322.4  269.42  5499.4  275.24    5528  277.76  5563.1  277.22
  5918.4  288.36  6031.6  289.93  6138.4  295.95  6181.3  295.28  6220.4  297.37
#Mann= 8 ,-1 , 0
  3950.7     .11       0  4183.6     .17       0  4201.8     .11       0
  4806.6     .15       0  4962.2     .11       0  4974.4     .07       0
  5024.4     .15       0  5232.6     .17       0
#XS Ineff= 2 , 0
       0                  5102.4       0  269.99
Permanent Ineff=
       F       F
Bank Sta=4974.4,5024.4
XS Rating Curve= 0 ,0
Exp/Cntr=0.3,0.1

Type RM Length L Ch R = 1 ,28713   ,498,498,498
BEGIN DESCRIPTION:
MCDONALD CREEK 55.0
END DESCRIPTION:
XS GIS Cut Line= 3
      3785569.82     10221645.49      3784940.06     10222376.27
      3784180.23     10223461.28
#Sta/Elev= 30
  4035.3  296.75  4174.9  287.78  4246.2  285.08  4317.5   280.2  4352.6  280.03
  4586.3  266.01  4657.6  263.37  4824.6  260.96  4913.2  261.58  4976.9  263.46
  4983.5  262.63  4990.1  254.48  5005.3  254.48  5005.8  254.98    5006  256.79
  5012.3  258.68  5033.2  262.07  5143.8  262.68  5408.1  267.44  5464.7  271.53
    5572  275.01  5586.8  276.82  5628.6  276.44  5744.6  280.87  5765.5  282.68
    5815  283.42  5988.7  287.38  6265.1  296.15  6312.1     297  6324.6  298.68
#Mann= 7 ,-1 , 0
  4035.3     .11       0  4824.6     .15       0  4983.5     .09       0
  5033.2     .15       0  5143.8     .17       0    5815     .11       0
  6265.1     .17       0
Bank Sta=4983.5,5033.2
XS Rating Curve= 0 ,0
Exp/Cntr=0.3,0.1

Type RM Length L Ch R = 1 ,28215   ,576,576,576
BEGIN DESCRIPTION:
MCDONALD CREEK 54.0
END DESCRIPTION:
XS GIS Cut Line= 3
      3785374.49      10221481.2      3784777.76     10221956.36
      3783637.04     10222634.17
#Sta/Elev= 30
  4237.2  301.53  4335.1  295.53  4419.9  288.42    4521  283.22  4597.7  276.73
  4674.6  272.16    4792  264.75  4811.6   263.7  4946.9  259.28  4982.1  261.91
  4988.5  259.06  4992.2  254.16  5007.4  254.16  5011.5  259.53    5024  261.27
  5085.3  261.27  5093.1  261.23  5225.4  260.97    5289  260.38  5353.8  262.85
  5411.7  264.45    5587   276.1    5624  277.19  5746.7  289.05    5778  289.54
  5799.4  292.11  5842.2  294.18  5965.4  297.74  6272.7  298.16  6326.9  299.65
#Mann= 12 ,-1 , 0
  4237.2     .11       0    4521     .17       0  4674.6     .11       0
    4792     .15       0  4811.6     .11       0  4946.9     .15       0
  4982.1     .09       0    5024     .15       0  5085.3     .11       0
  5093.1     .15       0  5225.4     .17       0  5353.8     .11       0
Bank Sta=4982.1,5024
XS Rating Curve= 0 ,0
Exp/Cntr=0.3,0.1

Type RM Length L Ch R = 1 ,27639   ,917,917,917
BEGIN DESCRIPTION:
MCDONALD CREEK 53.0
END DESCRIPTION:
XS GIS Cut Line= 3
      3785276.84     10221148.22      3784549.76     10221498.36
      3783576.46     10222484.55
#Sta/Elev= 30
    4193  305.63  4230.2  303.18  4278.1  300.17  4300.3  299.84  4396.4  292.81
  4532.1  287.84  4581.2  284.84  4732.6  272.39  4837.3   263.6    4877   262.2
  4891.1  262.99  4927.8  259.56    4973  260.83  4990.1  259.79  4995.6  257.77
  4998.3  253.24  5002.7  250.29  5017.9  250.29  5024.5  259.14  5038.6  260.95
    5198  258.98  5356.8  260.63  5420.5  264.05  5453.9  267.38  5597.2  278.77
  5788.2  286.39  5943.8  290.57  6056.9  292.13  6191.2  296.94  6385.6  301.37
#Mann= 9 ,-1 , 0
    4193     .11       0  4230.2     .17       0  4278.1     .11       0
  4581.2     .17       0  4732.6     .15       0  4990.1     .09       0
  5024.5     .15       0    5198     .17       0  5453.9     .11       0
Bank Sta=4990.1,5024.5
XS Rating Curve= 0 ,0
Exp/Cntr=0.3,0.1

Type RM Length L Ch R = 1 ,26722   ,499,499,499
BEGIN DESCRIPTION:
MCDONALD CREEK 51.0
END DESCRIPTION:
XS GIS Cut Line= 3
      3785250.21     10221054.99      3784086.64     10221108.44
      3783412.54     10222341.85
#Sta/Elev= 30
  3835.2  304.53  3987.7  297.94  4027.8  294.97  4127.9  290.13  4206.2  284.33
  4332.9  274.93  4431.9  266.87  4432.1  266.85  4530.9  261.16  4688.5  258.52
  4708.5   259.1  4728.9  257.86  4828.6  258.05  4908.7  256.29  4968.8  258.89
  4978.8  257.67  4989.2  250.98  5004.6  250.98  5024.4  253.95  5030.1  258.18
  5090.9  258.54  5127.8  257.21  5257.3  265.28    5569  273.92  5686.8  279.08
  5825.2  288.17  5914.7   292.4  6173.3  300.23  6254.9   301.2  6405.6   305.6
#Mann= 11 ,-1 , 0
  3835.2     .11       0  4206.2     .17       0  4332.9     .15       0
  4431.9     .11       0  4432.1     .15       0  4530.9     .11       0
  4728.9     .15       0  4978.8     .09       0  5030.1     .15       0
  5090.9     .17       0  5257.3     .11       0
Bank Sta=4978.8,5030.1
XS Rating Curve= 0 ,0
Exp/Cntr=0.3,0.1

Type RM Length L Ch R = 1 ,26223   ,497,497,497
BEGIN DESCRIPTION:
MCDONALD CREEK 50.0
END DESCRIPTION:
XS GIS Cut Line= 3
      3784513.26     10219953.93      3783758.63     10220816.93
      3783345.62     10222284.73
#Sta/Elev= 30
  3853.6  295.21  3947.4  286.83  4067.9   279.9  4110.7  275.13  4153.4  272.33
  4345.3  263.97  4556.8  257.15  4734.3  257.79  4785.7  256.53  4854.8  257.23
  4953.5   255.2    4982   257.7  4989.6   254.5  4991.7  250.91  5007.1  250.91
  5014.7  256.06  5020.6  257.14  5100.1  257.26  5167.2   258.3  5240.4  257.54
    5264  258.59  5274.4  260.17  5320.5   261.3  5440.6  267.38  5460.3  267.25
  5758.6  278.46  5804.2  281.79    5825  281.85  5978.4  290.07  6524.8  304.97
#Mann= 7 ,-1 , 0
  3853.6     .17       0  4345.3     .11       0  4785.7     .15       0
    4982     .09       0  5020.6     .15       0  5100.1     .17       0
  5320.5     .11       0
Bank Sta=4982,5020.6
XS Rating Curve= 0 ,0
Exp/Cntr=0.3,0.1

Type RM Length L Ch R = 1 ,25726   ,500,500,500
BEGIN DESCRIPTION:
MCDONALD CREEK 49.0
END DESCRIPTION:
XS GIS Cut Line= 3
      3783971.61      10219736.4      3783495.31     10220513.55
      3782475.42     10221521.18
#Sta/Elev= 30
  4088.5  296.64  4123.9  294.41  4334.7  273.93  4466.2  266.34  4516.2  265.44
  4587.5  261.52  4605.1  260.82  4729.2  257.53  4750.4  256.41  4856.9  256.48
  4887.8  254.58  4945.8  255.34  4973.6  252.67  4982.5  253.43  4988.4   249.9
  4995.7  247.93  5011.4  247.93  5017.7  255.42  5194.4  255.65  5215.7  254.36
  5374.3  255.72  5505.6  254.36  5577.3  257.05  5682.4  260.73  5774.3  267.08
  5809.7  268.03    6043  282.47  6163.2  287.51  6226.8  291.94  6433.7  298.64
#Mann= 8 ,-1 , 0
  4088.5     .17       0  4587.5     .11       0  4605.1     .17       0
  4729.2     .15       0  4945.8     .09       0  5017.7     .15       0
  5374.3     .17       0  5577.3     .11       0
#XS Ineff= 2 , 0
       0    4677   259.3               0
Permanent Ineff=
       F       F
Bank Sta=4945.8,5017.7
XS Rating Curve= 0 ,0
Exp/Cntr=0.3,0.1

Type RM Length L Ch R = 1 ,25226   ,498,498,498
BEGIN DESCRIPTION:
MCDONALD CREEK 48.0
END DESCRIPTION:
XS GIS Cut Line= 3
      3783873.91     10219674.28      3783070.91     10220319.82
      3782342.58     10221391.92
#Sta/Elev= 30
  3969.7  295.53    4007  290.89    4079  285.17  4192.6  278.34  4242.2  276.19
  4277.4  275.84  4320.6  272.95  4469.4  267.04    4519  266.12  4661.4  259.62
  4754.2  253.92  4895.7  253.55  4981.4  254.21  4995.8  249.25  4998.8  249.77
  5003.1  248.72  5018.8  248.72  5025.7   254.3  5182.9  254.04  5211.6  253.02
  5255.4  254.08    5315  253.11  5385.2  254.93  5400.1  254.49  5436.1  257.17
  5463.1  257.17  5540.1  260.93  5630.2  264.57  5759.4  271.41  6296.1  302.44
#Mann= 6 ,-1 , 0
  3969.7     .17       0  4895.7     .15       0  4981.4     .09       0
  5025.7     .15       0    5315     .17       0  5540.1     .11       0
Bank Sta=4981.4,5025.7
XS Rating Curve= 0 ,0
Exp/Cntr=0.3,0.1

Type RM Length L Ch R = 1 ,24728   ,499,499,499
BEGIN DESCRIPTION:
MCDONALD CREEK 47.0
END DESCRIPTION:
XS GIS Cut Line= 3
      3783842.86     10219612.11        3782978.     10219958.37
      3781734.05     10220775.28
#Sta/Elev= 30
  4068.4  294.29  4264.8   278.7  4612.1  267.51  4857.1  252.43  4892.4  249.93
  4970.1  252.27  4980.9  247.81  5031.2  251.59  5037.1  248.84  5052.2  249.37
    5060  252.34  5190.9  253.03    5212  248.93  5227.1  253.29  5398.8  252.72
    5640  258.97  5676.5  260.14  5745.3  263.74  5760.4  270.56  5766.4  269.41
  5775.5  273.09  5781.5  271.95  5797.7  275.51  5817.6  275.37  5847.8  270.42
  5918.8  269.99  5978.3  269.54  5998.4  272.74  6147.4  277.09  6488.2   292.8
#Mann= 10 ,-1 , 0
  4068.4     .17       0  4857.1     .15       0  4970.1     .09       0
    5060     .15       0    5640     .11       0  5676.5     .17       0
  5797.7     .11       0  5918.8     .17       0  5978.3     .11       0
  6147.4     .17       0
#XS Ineff= 2 , 0
       0                  5573.6       0  257.72
Permanent Ineff=
       F       F
Bank Sta=4970.1,5060
XS Rating Curve= 0 ,0
Exp/Cntr=0.3,0.1

Type RM Length L Ch R = 1 ,24229   ,496,496,496
BEGIN DESCRIPTION:
MCDONALD CREEK 46.0
END DESCRIPTION:
XS GIS Cut Line= 3
      3783811.76     10219394.58      3782908.49     10219487.17
      3781676.36     10219922.88
#Sta/Elev= 30
    4092  296.18  4203.1  284.38  4327.1   274.2  4600.3  261.43    4679  256.66
  4842.2  250.99  4920.2  249.17  4970.5  251.33  4980.5  251.38  4987.4  249.66
  5052.6  251.41  5056.3  248.09  5072.4  248.09  5074.9  250.21  5088.8  251.86
  5119.7  249.49  5299.8  250.74  5340.1  250.55  5361.6  248.96  5392.4  249.99
  5418.1  253.17  5531.8  259.26    5732  271.17  5859.8  278.36  5927.7  285.21
  5958.6  285.42    6046  290.33  6231.4  295.74  6251.7  297.47  6306.9  298.33
#Mann= 7 ,-1 , 0
    4092     .17       0  4842.2     .15       0  5052.6     .09       0
  5088.8     .15       0  5392.4     .11       0  5531.8     .17       0
    5732     .11       0
Bank Sta=5052.6,5088.8
XS Rating Curve= 0 ,0
Exp/Cntr=0.3,0.1

Type RM Length L Ch R = 1 ,23733   ,499,499,499
BEGIN DESCRIPTION:
MCDONALD CREEK 45.0
END DESCRIPTION:
XS GIS Cut Line= 3
      3783802.87     10218999.46      3782808.25     10219018.03
      3781596.42     10219483.37
#Sta/Elev= 30
  4005.2  296.42  4180.3  278.23  4380.3  264.27  4660.3   250.3  4749.9  249.15
  4920.4   247.8  4980.4  248.88  4989.6  242.49  5005.8  242.49  5011.1  246.32
  5019.5   249.1  5079.5  247.76  5118.3  248.93  5128.8  248.64  5139.7   245.9
  5164.2   248.8  5268.2  248.48  5328.2  251.98  5358.2  252.39  5467.6   260.4
  5497.6  261.53  5552.3  266.31  5582.3  266.98  5606.9  269.76    5637  269.46
  5643.1  270.58  5739.5  274.38    5861  277.48  5975.7  282.54  6298.1  291.13
#Mann= 5 ,-1 , 0
  4005.2     .17       0  4749.9     .15       0  4980.4     .09       0
  5019.5     .15       0  5268.2     .11       0
#XS Ineff= 2 , 0
       0                  5352.9       0  252.85
Permanent Ineff=
       F       F
Bank Sta=4980.4,5019.5
XS Rating Curve= 0 ,0
Exp/Cntr=0.3,0.1

Type RM Length L Ch R = 1 ,23234   ,475,475,475
BEGIN DESCRIPTION:
MCDONALD CREEK 44.0
END DESCRIPTION:
XS GIS Cut Line= 3
      3783793.97       10218702.      3782678.35     10218555.49
      3781463.26     10219221.41
#Sta/Elev= 30
  3874.8  289.62  4007.5  277.95  4203.7  265.07  4395.4  255.49  4566.8  250.12
  4716.3  248.24  4849.2  246.17  4929.9   246.7  4950.1  245.48  4980.3  247.16
  4987.4  241.39  5003.6  241.39  5019.8   245.9  5034.8  246.61  5085.3  245.26
  5131.2   246.6  5226.5  248.22  5460.7  258.42  5482.5  262.62  5498.6  268.58
  5504.3  269.09  5513.7  268.81  5520.4  266.31  5542.2     264    5874  264.51
  5917.6  266.78  5955.5  270.72  6072.5  276.47  6255.1  284.07  6385.6  287.13
#Mann= 6 ,-1 , 0
  3874.8     .17       0  4007.5     .11       0  4716.3     .15       0
  4980.3     .09       0  5034.8     .15       0  5131.2     .11       0
Bank Sta=4980.3,5034.8
XS Rating Curve= 0 ,0
Exp/Cntr=0.3,0.1

Type RM Length L Ch R = 1 ,22759   ,941,941,941
BEGIN DESCRIPTION:
MCDONALD CREEK 42.0
END DESCRIPTION:
XS GIS Cut Line= 3
      3783474.34     10217645.39      3782515.66     10218207.07
      3781420.19     10219087.15
#Sta/Elev= 30
  3888.9   284.6  4030.3  275.07  4165.8  268.05  4206.5  265.95  4336.8  257.34
  4440.6  254.73  4568.6  249.68  4685.9  248.04  4781.7   242.2  4797.4  246.01
  4846.8   246.9  4856.1  243.32  4861.9   246.5  4868.8  240.36  4869.3  239.86
  4886.3  240.36  4893.2  246.92    4899  248.21  4927.9  247.13  4951.1  248.78
 4975.59  246.87    4999  241.22  5036.2  246.73  5172.2  245.58  5300.2  247.75
  5605.8  261.34    5677  266.61  5698.6  265.55  5818.6  270.42  6405.2  285.91
#Mann= 9 ,-1 , 0
  3888.9     .17       0  4030.3     .11       0  4165.8     .17       0
  4206.5     .11       0  4440.6     .15       0  4868.8     .09       0
  4886.3     .15       0 4975.59     .09       0  5036.2     .15       0
Bank Sta=4975.59,5036.2
XS Rating Curve= 0 ,0
Exp/Cntr=0.3,0.1

Type RM Length L Ch R = 1 ,21818   ,576,576,576
BEGIN DESCRIPTION:
MCDONALD CREEK 41.0
END DESCRIPTION:
XS GIS Cut Line= 3
      3783185.82     10217232.47      3782485.46     10217714.12
      3781374.42     10219039.42
#Sta/Elev= 30
    4150  286.83  4268.9  278.52  4313.3  276.86  4355.2  272.17  4499.5  261.87
  4621.1  256.25  4671.8  251.42  4742.4  249.49  4809.1  246.38  4937.7  243.62
  4973.5  245.23  4982.3  245.01    4995  241.56  5011.6  241.56  5017.6  244.52
  5031.9  245.16  5146.6  244.46  5422.2  243.75  5455.8  244.95  5514.6  247.08
  5570.6  251.81  5642.1  254.69  5648.6  253.56  5656.4  255.75  5662.9  254.77
  5670.7  257.91  5691.5  260.68  5968.7  267.42  6202.8  275.34  6729.4  285.22
#Mann= 6 ,-1 , 0
    4150     .17       0  4742.4     .15       0  4973.5     .09       0
  5031.9     .15       0  5146.6     .17       0  5455.8     .11       0
Bank Sta=4973.5,5031.9
XS Rating Curve= 0 ,0
Exp/Cntr=0.3,0.1

Type RM Length L Ch R = 1 ,21242   ,497,497,497
BEGIN DESCRIPTION:
MCDONALD CREEK 40.0
END DESCRIPTION:
XS GIS Cut Line= 3
      3783017.86     10216961.07      3782401.06     10217221.19
      3780544.22      10218342.4
#Sta/Elev= 30
  4330.6  291.14  4384.9  288.08  4529.2  272.43  4574.9   267.7  4632.7  264.28
  4638.1  263.73  4651.5  261.84  4680.7  261.39    4747  254.68  4833.8     249
    4895  247.81  4957.9  242.37  5168.7  242.67  5255.5  240.58  5337.5  242.79
  5500.9   246.7  5591.8   250.3  5607.3  252.82  5665.5  255.77  5941.1  257.32
  6152.6  265.64  6168.1  268.24  6189.5  267.51  6276.4  270.53  6530.4  275.25
  6577.4  276.38  6655.3  278.91  6909.5  276.28  7114.5  280.01  7169.1  281.58
#Mann= 12 ,-1 , 0
  4330.6     .17       0  4529.2     .11       0  4632.7     .17       0
  4638.1     .11       0    4747     .15       0  5168.7     .09       0
  5337.5     .15       0  5500.9     .17       0  6276.4     .15       0
  6530.4     .17       0  6577.4     .15       0  7114.5     .11       0
Bank Sta=5168.7,5337.5
XS Rating Curve= 0 ,0
Exp/Cntr=0.3,0.1

Type RM Length L Ch R = 1 ,20745   ,470,470,470
BEGIN DESCRIPTION:
MCDONALD CREEK 39.0
END DESCRIPTION:
XS GIS Cut Line= 3
      3782990.49     10216908.41       3782272.3     10216866.76
      3780517.58     10218302.44
#Sta/Elev= 30
  4280.6  290.38  4313.3  288.03  4491.1  268.09  4628.5  257.53  4727.1  250.14
  4774.1  246.32  4974.4  241.97  5006.1  238.32  5011.6  235.75  5028.2  235.75
  5034.3   240.4  5042.2  242.32    5063  240.84  5176.4   238.8  5212.5  242.02
  5265.2  242.54  5510.2  249.09  5532.4  252.15  5567.6  250.47  5631.5  254.99
  5872.7   257.5  6099.8  263.89  6150.5  266.51    6200  266.45    6427  273.28
  6634.4  274.98  6664.4  274.79  7003.2  275.17  7198.2  279.27  7267.2   281.1
#Mann= 10 ,-1 , 0
  4280.6     .17       0  4628.5     .11       0  4727.1     .15       0
  4974.4     .09       0  5042.2     .15       0  5265.2     .17       0
  6099.8     .15       0  6634.4     .17       0  6664.4     .15       0
  7198.2     .11       0
#XS Ineff= 2 , 0
       0                  5439.8       0  247.11
Permanent Ineff=
       F       F
Bank Sta=4974.4,5042.2
XS Rating Curve= 0 ,0
Exp/Cntr=0.3,0.1

Type RM Length L Ch R = 1 ,20275   ,500,500,500
BEGIN DESCRIPTION:
MCDONALD CREEK 38.0
END DESCRIPTION:
XS GIS Cut Line= 3
      3782635.29      10215878.4      3782069.14     10216604.58
      3780478.57     10218257.07
#Sta/Elev= 30
  4079.2  281.88  4521.2   249.5  4570.9  247.83  4606.2  244.62  4706.6  242.53
  4883.9  239.63  4962.6  240.87  4977.1  240.23    4983  235.04  5000.1  235.04
  5005.6  239.58  5012.5  240.51  5175.4  239.93  5217.5  243.86  5223.8  243.46
  5387.3  250.42    5437  250.12  5862.9  257.87    5932     259  5995.5  262.06
    6137  263.46    6215  266.17  6221.9   265.3  6229.1  266.41  6264.4     266
  6429.3  269.19  6616.8  270.82    6915  272.16  7197.3  278.15  7293.6  281.24
#Mann= 9 ,-1 , 0
  4079.2     .17       0  4706.6     .15       0  4962.6     .09       0
  5012.5     .15       0  5223.8     .17       0  5862.9     .15       0
  6429.3     .17       0  6616.8     .15       0  7197.3     .11       0
#XS Ineff= 2 , 0
       0                  5302.4       0  247.48
Permanent Ineff=
       F       F
Bank Sta=4962.6,5012.5
XS Rating Curve= 0 ,0
Exp/Cntr=0.3,0.1

Type RM Length L Ch R = 1 ,19775   ,497,497,497
BEGIN DESCRIPTION:
MCDONALD CREEK 37.0
END DESCRIPTION:
XS GIS Cut Line= 3
      3782502.12      10215767.4      3781732.02     10216300.82
      3780242.55     10217205.72
#Sta/Elev= 30
  4063.2  286.79  4213.6  275.22  4479.1  250.21  4535.9  246.19  4550.8  246.55
    4663  241.06  4750.7  238.84  4881.8  238.33  4980.7  239.64  4986.8  234.74
  5003.9  234.74  5005.1  237.59  5016.6  239.28  5075.1  238.76  5146.7  240.71
  5279.8  243.18  5301.1  241.31  5344.2  244.74  5417.4  245.77  5448.4  244.09
  5484.6  246.39  5578.2  247.97    5929  260.44  6299.2  270.76  6430.9  275.33
  6516.2  280.12  6553.1  279.53    6584  282.02  6589.9  280.89  6742.8  284.37
#Mann= 5 ,-1 , 0
  4063.2     .17       0    4663     .15       0  4980.7     .09       0
  5016.6     .15       0  5146.7     .17       0
#XS Ineff= 4 ,-1
  4542.8  4529.8  246.61  5359.3  5426.1  245.09  5496.9  5533.7  246.59
  5426.1  5496.9  245.86
Permanent Ineff=
       F       F       F       F
Bank Sta=4980.7,5016.6
XS Rating Curve= 0 ,0
Exp/Cntr=0.3,0.1

Type RM Length L Ch R = 1 ,19278   ,500,500,500
BEGIN DESCRIPTION:
MCDONALD CREEK 36.0
END DESCRIPTION:
XS GIS Cut Line= 3
      3782484.35     10215687.51      3781396.39     10215984.99
      3780189.06      10217121.5
#Sta/Elev= 30
  3872.1  287.44  3944.3  285.14  4166.9  267.06  4500.9  250.72    4588  244.47
  4687.5  240.84  4741.6  240.84  4776.1  235.68  4785.6  240.31  4801.5  242.07
  4863.7  239.45    4957  238.68  4969.4  237.28  4977.7  233.03  4979.4  229.51
  4996.9  229.51  5003.2  235.54  5010.5  238.21  5080.9  235.19  5114.9  237.85
  5484.3  246.97  5519.9  245.06  5604.4  251.83  5823.7  259.99  5873.5  259.91
  5930.2  263.91  5986.8  264.21  6177.8   270.7  6488.9  283.29  6658.1  285.35
#Mann= 5 ,-1 , 0
  3872.1     .17       0  4785.6     .15       0    4957     .09       0
  5010.5     .15       0  5114.9     .17       0
#XS Ineff= 2 , 0
       0                  5463.3       0  246.56
Permanent Ineff=
       F       F
Bank Sta=4957,5010.5
XS Rating Curve= 0 ,0
Exp/Cntr=0.3,0.1

Type RM Length L Ch R = 1 ,18778   ,498,498,498
BEGIN DESCRIPTION:
MCDONALD CREEK 35.0
END DESCRIPTION:
XS GIS Cut Line= 3
       3781951.6     10214954.96      3780959.06     10215838.01
      3780132.11     10217062.65
#Sta/Elev= 30
  3671.5  276.27  3806.1   275.4  4195.8  265.28  4316.2  259.35  4485.9  246.58
    4617  239.66  4691.6  238.14  4712.5   235.8  4747.7  237.28  4769.4  235.95
  4988.5  237.83    4996  234.69  4998.5  230.96  5001.7  229.21  5019.2  229.21
  5025.4   233.7  5052.4  238.07  5073.8   239.3  5184.2  241.64  5256.2  246.92
  5570.9  259.73  5594.8   262.4  5651.8  261.79  5765.8  266.28  5810.7  266.32
  5831.7  268.24  5932.8  270.52  6083.4  277.72  6320.3  286.31  6477.7  286.97
#Mann= 5 ,-1 , 0
  3671.5     .17       0    4617     .15       0  4988.5     .09       0
  5052.4     .15       0  5073.8     .17       0
Bank Sta=4988.5,5052.4
XS Rating Curve= 0 ,0
Exp/Cntr=0.3,0.1

Type RM Length L Ch R = 1 ,18280   ,499,499,499
BEGIN DESCRIPTION:
MCDONALD CREEK 34.0
END DESCRIPTION:
XS GIS Cut Line= 3
      3781880.57     10214892.81      3780888.18     10215435.95
      3780082.68     10216974.67
#Sta/Elev= 30
  3868.7  278.17  4031.4   276.6  4474.9  253.72    4533  252.24    4590   247.8
  4627.6  247.45  4760.2  239.16  4886.4  234.95  4915.9  236.77    4932  236.06
  4937.7  232.72  4943.4   236.3  4959.5  236.42  4975.6  232.55  4981.3  234.29
  5002.7  228.89  5020.2  228.89  5027.9  236.35  5033.5  236.77  5084.8  235.35
  5154.2  236.92  5165.9  234.87  5182.4  234.94    5381  245.98  5485.7  247.16
  5612.4  252.58  5640.1  255.27  6026.1  264.65    6507  283.35  6736.8  289.21
#Mann= 5 ,-1 , 0
  3868.7     .17       0  4760.2     .15       0  4959.5     .09       0
  5033.5     .15       0  5154.2     .17       0
#XS Ineff= 2 , 0
       0  4709.2  243.16               0
Permanent Ineff=
       F       F
Bank Sta=4959.5,5033.5
XS Rating Curve= 0 ,0
Exp/Cntr=0.3,0.1

Type RM Length L Ch R = 1 ,17781   ,498,498,498
BEGIN DESCRIPTION:
MCDONALD CREEK 33.0
END DESCRIPTION:
XS GIS Cut Line= 3
      3781853.92     10214830.67       3781033.3     10215052.22
      3779519.13     10215656.26
#Sta/Elev= 30
    4150  278.59  4365.6  274.81    4581  265.88  4684.5  259.35  4818.5  248.58
  4823.7  246.53  4839.9  246.35  4863.6  243.14  4938.2  239.82  4984.9  234.82
  4996.7  227.72  5014.2  227.72  5014.7  228.22  5016.6  235.39  5064.7  237.17
  5095.6  236.18  5210.4  234.33  5393.5  235.32  5645.2  240.17    5717   239.3
  5932.6  245.19  6157.9  255.16  6190.2  254.25  6233.2  257.77    6256  256.23
  6304.5  262.53    6325  263.56  6525.5  277.79  6588.5  284.92  6630.2  287.19
#Mann= 6 ,-1 , 0
    4150     .17       0  4984.9     .09       0  5016.6     .17       0
  5095.6     .15       0  5645.2     .11       0    6325     .17       0
Bank Sta=4984.9,5016.6
XS Rating Curve= 0 ,0
Exp/Cntr=0.3,0.1
