--- STEWART CREEK NORTH.prj (project) ---

Proj Title=STEWART CREEK NORTH Base Level Engineering
Current Plan=p01
Default Exp/Contr=0.3,0.1
English Units
Geom File=g01
Flow File=f01
Plan File=p01
Y Axis Title=Elevation
X Axis Title(PF)=Main Channel Distance
X Axis Title(XS)=Station
BEGIN DESCRIPTION:
STEWART CREEK NORTH
END DESCRIPTION:
DSS File=dss
DSS Export Rating Curves= 0
DSS Export Rating Curve Sorted= 0
DSS Export Volume Flow Curves= 0
DXF OffsetX= 0
DXF OffsetY= 0
DXF ScaleX= 1
DXF ScaleY= 10

--- STEWART CREEK NORTH.p01 (plan) ---

Plan Title=Multiple Run
Program Version=4.10
Short Identifier=Multiple Run
Geom File=g01
Flow File=f01
Subcritical Flow
K Sum by GR= 0
Std Step Tol= 0.01
Critical Tol= 0.01
Num of Std Step Trials= 20
Max Error Tol= 0.3
Flow Tol Ratio= 0.001
Split Flow NTrial= 30
Split Flow Tol= 0.02
Split Flow Ratio= 0.02
Log Output Level= 0
Friction Slope Method= 1
Unsteady Friction Slope Method= 2
Unsteady Bridges Friction Slope Method= 1
Parabolic Critical Depth
Global Vel Dist= 1 , 1 , 1
Global Log Level= 0
CheckData=True
Encroach Param=-1 ,0,0, 0
BEGIN DESCRIPTION:
Multiple Run
END DESCRIPTION:
Computation Interval=1HOUR
Output Interval=1HOUR
Run HTab= 0
Run UNet= 0
Run PostProcess= 0
Run WQNet= 0
UNET Theta= 1
UNET Theta Warmup= 1
UNET ZTol= 0.02
UNET ZSATol= 0.05
UNET MxIter= 20
UNET MaxInSteps= 0
UNET DtIC= 0
UNET DtMin= 0
UNET MaxCRTS= 20
UNET WFStab= 2
UNET SFStab= 1
UNET WFX= 1
UNET SFX= 1
UNET DSS MLevel= 4
UNET DZMax Abort= 100
UNET Convert EG Bridges= 0
UNET Use Existing IB Tables=-1
UNET Froude Reduction=False
UNET Froude Limit= 1
UNET Froude Power= 10
UNET Time Slicing=0,0, 5
UNET Junction Losses=0
Instantaneous Interval=1HOUR
DSS File=dss
Write IC File= 0
Write IC File at Sim End=0
Echo Input=False
Echo Parameters=False
Echo Output=False
Write Detailed= 0
WQ AD Non Conservative
WQ ULTIMATE=-1
WQ Max Comp Step=1HOUR
WQ Output Interval=15MIN
WQ Output Selected Increments= 0
WQ Output face flow=0
WQ Output face velocity=0
WQ Output face area=0
WQ Output face dispersion=0
WQ Output cell volume=0
WQ Output cell surface area=0
WQ Output cell continuity=0
WQ Output cumulative cell continuity=0
WQ Output face conc=0
WQ Output face dconc_dx=0
WQ Output face courant=0
WQ Output face peclet=0
WQ Output face adv mass=0
WQ Output face disp mass=0
WQ Output cell mass=0
WQ Output cell source sink temp=0
WQ Output cell source sink nsm=0
WQ Output MaxMinRange=-1
WQ Daily Max Min Mean=-1
WQ Daily Range=0
WQ Daily Time=0
WQ Create Restart=0
WQ Fixed Restart=0
WQ System Summary=0
WQ Use Fixed Temperature=0
Sorting and Armoring Iterations= 10
XS Update Threshold= 0.02
Hydraulics Update Threshold= 0.02
Energy Slope Method= 1
Volume Change Method= 0
XS Weighting Method= 0
Number of US Weighted Cross Sections= 1
Number of DS Weighted Cross Sections= 1
Upstream XS Weight=0.25
Main XS Weight=0.5
Downstream XS Weight=0.25
Number of DS XS's Weighted with US Boundary= 1
Upstream Boundary Weight= 1
Weight of XSs Associated with US Boundary= 0
Number of US XS's Weighted with DS Boundary= 1
Downstream Boundary Weight= 0.5
Weight of XSs Associated with DS Boundary= 0.5
Sediment Output Level= 4
Mass or Volume Output= 0
Output Increment Type= 1
Profile and TS Output Increment= 10
XS Output Flag= 0
XS Output Increment= 10
Disregard all LS=0
Disregard all Conn=0
Disregard all Breaches=0
Disregard all Pumps=0

--- STEWART CREEK NORTH.f01 (steady flow) ---

Flow Title=Multiple
Program Version=4.10
Number of Profiles= 7
Profile Names=10-year,25-year,50-year,1pct_min,100-year,1pct_plu,500-year
River Rch & RM=STEWART CREEK NO,Reach-1         ,45625
     256     329     430     186     562    1697     984
River Rch & RM=STEWART CREEK NO,Reach-1         ,45000
     662     905    1232     552    1668    5037    3160
River Rch & RM=STEWART CREEK NO,Reach-1         ,40756
    1200    1686    2336    1062    3207    9685    6257
River Rch & RM=STEWART CREEK NO,Reach-1         ,38500
    1552    2203    3073    1406    4245   12820    8385
River Rch & RM=STEWART CREEK NO,Reach-1         ,34500
    1823    2601    3639    1669    5039   15218   10002
River Rch & RM=STEWART CREEK NO,Reach-1         ,31500
    1944    2764    3858    1764    5326   16084   10507
River Rch & RM=STEWART CREEK NO,Reach-1         ,24000
    1977    2801    3899    1776    5363   16196   10511
River Rch & RM=STEWART CREEK NO,Reach-1         ,21000
    3611    5172    7251    3319   10023   30269   19830
River Rch & RM=STEWART CREEK NO,Reach-1         ,17000
    3562    5063    7060    3214    9706   29312   18987
River Rch & RM=STEWART CREEK NO,Reach-1         ,14000
    4452    6377    8940    4090   12351   37299   24400
River Rch & RM=STEWART CREEK NO,Reach-1         ,10500
    4508    6457    9053    4141   12507   37771   24704
River Rch & RM=STEWART CREEK NO,Reach-1         ,10000
    4481    6406    8967    4096   12370   37357   24357
River Rch & RM=STEWART CREEK NO,Reach-1         ,8000
    4656    6668    9348    4276   12913   38997   25497
River Rch & RM=STEWART CREEK NO,Reach-1         ,3500
    4206    5952    8272    3751   11327   34207   21973
River Rch & RM=STEWART CREEK NO,Reach-1         ,1500
    4303    6096    8480    3847   11619   35089   22575
Boundary for River Rch & Prof#=STEWART CREEK NO,Reach-1         , 1
Up Type= 0
Dn Type= 3
Dn Slope=0.005
Boundary for River Rch & Prof#=STEWART CREEK NO,Reach-1         , 2
Up Type= 0
Dn Type= 3
Dn Slope=0.005
Boundary for River Rch & Prof#=STEWART CREEK NO,Reach-1         , 3
Up Type= 0
Dn Type= 3
Dn Slope=0.005
Boundary for River Rch & Prof#=STEWART CREEK NO,Reach-1         , 4
Up Type= 0
Dn Type= 3
Dn Slope=0.005
Boundary for River Rch & Prof#=STEWART CREEK NO,Reach-1         , 5
Up Type= 0
Dn Type= 3
Dn Slope=0.005
Boundary for River Rch & Prof#=STEWART CREEK NO,Reach-1         , 6
Up Type= 0
Dn Type= 3
Dn Slope=0.005
Boundary for River Rch & Prof#=STEWART CREEK NO,Reach-1         , 7
Up Type= 0
Dn Type= 3
Dn Slope=0.005
DSS Import GetInterval= 0
DSS Import GetPeak= 0
DSS Import FillOption= 0

--- STEWART CREEK NORTH.g01 (geometry) ---

Geom Title=Existing Conditions
Program Version=4.10

River Reach=STEWART CREEK NO,Reach-1
Reach XY= 30
      3757927.96     10133938.96      3759362.35     10134065.52
      3759537.28     10133726.67      3760570.15     10134103.75
      3760671.21     10133776.89      3761150.26     10134270.34
      3761089.71     10134512.55      3762866.21     10134480.31
      3763917.69     10135006.06      3764049.07     10135524.82
      3764892.15     10135901.56      3765067.36     10136214.26
      3765716.42     10136254.36      3766011.26     10137214.56
      3767284.42     10137382.43      3767733.39     10137812.39
      3768598.68     10138085.62      3769111.02     10137637.19
      3770508.14     10137829.53      3771045.77     10137443.09
      3773362.85     10136858.39      3775728.88     10137109.84
      3776155.64     10136809.87      3777676.61     10136683.48
       3779028.6     10136229.79      3780650.62     10134691.08
      3782343.05     10133791.66       3784764.1     10133516.54
      3787880.85     10133819.76      3795967.33     10134043.51

Type RM Length L Ch R = 1 ,45625   ,106,106,106
BEGIN DESCRIPTION:
STEWART CREEK NORTH 91.5
END DESCRIPTION:
XS GIS Cut Line= 3
      3758083.15     10134577.09      3758083.31     10133942.09
      3758085.56      10133555.5
#Sta/Elev= 30
    4365  274.16    4411  275.92    4481  276.17    4541  277.53    4561  277.12
    4571  276.15    4581  276.67    4611  276.01    4651  276.12    4671  275.19
    4751  273.52    4791  273.84    4801  273.07    4811  273.55    4941  269.84
    4971  269.97    5003   268.2    5009  267.38  5009.3  266.88    5071  269.79
    5081  269.67    5101  271.17    5141  271.18    5231  274.58    5251  274.69
    5311  279.77    5341  279.99    5351  281.44    5381  281.81  5386.6  282.37
#Mann= 3 , 0 , 0
    4365     .11       0    4971     .07       0    5071     .11       0
Bank Sta=4971,5071
XS Rating Curve= 0 ,0
Exp/Cntr=0.3,0.1

Type RM Length L Ch R = 1 ,45519   ,519,519,519
BEGIN DESCRIPTION:
STEWART CREEK NORTH 91.0
END DESCRIPTION:
XS GIS Cut Line= 3
       3758179.8     10134593.96       3758178.8     10133987.56
      3758201.55     10133538.03
#Sta/Elev= 30
  4393.6  277.37  4416.5  275.78  4436.5  272.37  4528.3   273.3  4596.5  273.67
  4606.5  274.41  4621.3  273.82  4756.5  272.78  4786.5  270.74  4806.5  271.21
  4846.5  269.33  4986.5  265.79    4994  264.66  5026.5  266.71  5046.5  266.12
  5066.6  267.57  5075.9  269.45  5086.6   270.6  5116.6  271.36  5136.7  270.14
  5166.7  270.26  5176.7  271.38  5274.9  273.61  5279.9  275.65  5286.9  275.97
  5326.9   274.8  5346.9  277.05    5397  277.66    5417  279.31  5450.1  280.04
#Mann= 5 ,-1 , 0
  4393.6     .11       0  4528.3     .15       0  4621.3     .11       0
  4846.5     .07       0  5075.9     .11       0
Bank Sta=4846.5,5075.9
XS Rating Curve= 0 ,0
Exp/Cntr=0.3,0.1

Type RM Length L Ch R = 1 ,45000   ,500,500,500
BEGIN DESCRIPTION:
STEWART CREEK NORTH 90.0
END DESCRIPTION:
XS GIS Cut Line= 3
      3758823.21     10134454.92      3758630.62     10134146.16
      3758530.28     10133652.04
#Sta/Elev= 30
  4636.1  276.05  4678.2   275.8  4782.1  272.63  4802.6  271.42  4888.2  270.38
  4911.7  269.13  4918.9  268.72  4924.8  266.54  4940.1  265.37  4947.1  263.36
  4968.6  258.81  4968.9  258.31  5005.2   260.1    5040  260.36  5066.4  262.91
  5076.6  262.77    5097  263.64  5107.2  265.19  5117.4  267.51  5127.6  268.54
  5141.2  268.76    5148  269.53  5165.6  269.45  5242.5   270.3  5301.1  271.92
  5311.3  271.21  5343.8  273.54  5403.1  275.12  5413.4   274.8  5504.2  277.01
#Mann= 6 ,-1 , 0
  4636.1     .11       0  4802.6     .15       0  4947.1     .09       0
  5066.4     .15       0  5165.6    .125       0  5403.1     .11       0
Bank Sta=4947.1,5066.4
XS Rating Curve= 0 ,0
Exp/Cntr=0.3,0.1

Type RM Length L Ch R = 1 ,44500   ,500,500,500
BEGIN DESCRIPTION:
STEWART CREEK NORTH 89.0
END DESCRIPTION:
XS GIS Cut Line= 3
      3758888.35     10134435.39      3758954.06     10133951.64
      3758693.02     10133606.42
#Sta/Elev= 30
  4511.8  276.33  4586.8  274.34  4649.7  274.37  4778.5  271.58  4818.9  268.27
  4838.3  261.95  4849.2  260.36  4929.9  259.36  4950.1   256.5  4980.4  255.98
  5002.7   253.3  5012.8  255.36    5019  254.65  5033.6  257.86  5039.9  256.88
  5048.2  259.01  5054.4  258.63  5062.7  260.78    5069  258.84  5083.5   262.4
  5089.8  261.64  5107.2   263.5  5183.4  267.98  5247.9   269.2  5262.5  270.95
  5276.5  270.36  5376.8  273.09  5383.2  272.33  5402.3  273.76  5432.8  274.54
#Mann= 6 ,-1 , 0
  4511.8     .11       0  4649.7     .15       0  4929.9     .09       0
  5048.2     .15       0  5107.2     .17       0  5402.3     .11       0
Bank Sta=4929.9,5048.2
XS Rating Curve= 0 ,0
Exp/Cntr=0.3,0.1

Type RM Length L Ch R = 1 ,44000   ,500,500,500
BEGIN DESCRIPTION:
STEWART CREEK NORTH 88.0
END DESCRIPTION:
XS GIS Cut Line= 4
      3759085.83     10134413.69       3759219.8     10133964.96
      3759218.09     10133939.44      3758719.04     10133586.88
#Sta/Elev= 30
  4531.7  277.13  4722.3  272.62  4734.5  271.06  4752.9  266.77  4762.4  264.72
  4872.2  260.61  4905.4  255.64  4920.6  257.74    4931  257.47  4938.5  255.59
  4943.7  256.25  4951.9  253.96  4962.3  252.82  4993.6  252.06  4997.7  250.74
  5031.7  255.51  5046.5  252.75  5061.3   252.1  5067.4  254.04  5082.2  255.21
  5088.3  256.65  5111.6  257.42  5183.2  258.24  5303.1  263.27  5325.9  265.17
  5332.1  264.24  5346.9  264.84  5376.4  267.29  5635.1  273.37  5636.6  273.37
#Mann= 6 ,-1 , 0
  4531.7     .11       0  4752.9     .17       0    4931     .09       0
  5111.6     .15       0  5303.1     .17       0  5635.1     .11       0
Bank Sta=4931,5111.6
XS Rating Curve= 0 ,0
Exp/Cntr=0.3,0.1

Type RM Length L Ch R = 1 ,43500   ,500,500,500
BEGIN DESCRIPTION:
STEWART CREEK NORTH 87.0
END DESCRIPTION:
XS GIS Cut Line= 4
      3759604.48     10134263.95      3759456.81     10133836.14
      3759441.17     10133830.21      3758838.42     10133593.41
#Sta/Elev= 30
  4530.7  269.55  4568.5  268.79  4629.7  265.53  4693.3  262.98  4776.3  262.87
  4787.6  261.03  4798.2  261.53  4833.5   258.9  4925.2  256.34  4937.6  254.45
  4963.5  252.35  4968.8  250.26  4985.5   250.1  4991.1  247.62  5004.5  248.36
  5010.1  249.91  5015.5  248.46  5025.1  250.33  5046.5  251.13  5069.7   254.7
  5118.5  255.89  5232.3  256.08  5262.1  258.16  5340.7  259.67  5389.6  263.01
  5478.1  264.99  5540.8  266.98    5563  268.78    5582  267.71  5647.6  270.09
#Mann= 6 ,-1 , 0
  4530.7     .11       0  4629.7     .17       0  4833.5     .15       0
  4937.6     .09       0  5069.7     .15       0  5478.1     .17       0
Bank Sta=4937.6,5069.7
XS Rating Curve= 0 ,0
Exp/Cntr=0.3,0.1

Type RM Length L Ch R = 1 ,43000   ,500,500,500
BEGIN DESCRIPTION:
STEWART CREEK NORTH 86.0
END DESCRIPTION:
XS GIS Cut Line= 3
       3759626.2      10134259.6      3759720.22      10133866.8
      3759726.01     10133478.44
#Sta/Elev= 30
  4596.1  268.89  4650.5  266.65  4706.6   263.5  4711.7  264.23  4728.3  264.21
  4748.6   261.7  4753.8  262.34  4759.1   261.5  4837.8  257.77    4843  258.55
  4851.7  257.73  4872.2  257.62  4908.5  252.73  4921.9  250.63  4927.1  251.17
  4933.9  249.49  4954.5  250.37  4969.1  249.52  4985.3   250.2  4993.5  245.53
    5000  246.03  5005.7  248.68  5015.7  249.77  5075.7  252.79  5095.7  252.07
  5178.9  253.82  5195.7  253.96  5315.8  259.49  5345.8  262.57  5388.4  263.96
#Mann= 5 ,-1 , 0
  4596.1     .11       0  4650.5     .17       0  4908.5     .09       0
  5075.7     .15       0  5178.9     .11       0
Bank Sta=4908.5,5075.7
XS Rating Curve= 0 ,0
Exp/Cntr=0.3,0.1

Type RM Length L Ch R = 1 ,42500   ,500,500,500
BEGIN DESCRIPTION:
STEWART CREEK NORTH 85.0
END DESCRIPTION:
XS GIS Cut Line= 3
      3759884.44     10134261.79      3760016.47     10133939.81
      3759830.18     10133467.53
#Sta/Elev= 30
    4652   264.9    4701  263.85  4763.2  261.35  4783.7  260.58  4814.9  258.28
  4837.1  257.82  4914.5  254.24  4933.1  252.14  4944.6  249.39  4962.5  249.11
  4967.9  247.41    5002  245.58  5005.2  244.38  5008.7  244.38  5012.3     246
  5036.7  246.02  5042.1  246.73  5084.6  246.19  5096.2  247.21  5106.1   247.1
  5120.6  248.57  5127.6  250.36  5138.4  250.49  5159.9  249.08  5169.3  250.05
  5198.5  250.65  5321.1  253.67  5385.6  257.87  5391.2  258.85  5507.7  264.34
#Mann= 5 ,-1 , 0
    4652     .11       0  4763.2     .17       0  4962.5     .09       0
  5120.6     .15       0  5198.5     .11       0
Bank Sta=4962.5,5120.6
XS Rating Curve= 0 ,0
Exp/Cntr=0.3,0.1

Type RM Length L Ch R = 1 ,42000   ,459,459,459
BEGIN DESCRIPTION:
STEWART CREEK NORTH 84.0
END DESCRIPTION:
XS GIS Cut Line= 4
      3760181.74     10134281.37      3760280.77     10133889.08
      3760276.69     10133875.64      3759952.36      10133446.7
#Sta/Elev= 30
  4595.4  258.74  4641.5  257.95  4657.6  258.45  4718.4   256.7  4740.1  257.08
    4771  254.89  4800.5  254.44  4851.1  251.45  4863.9  250.32  4894.8  250.15
  4905.1  248.68  4915.4  246.92  4928.8   247.6  4946.4  243.27  4964.7  246.09
  4969.9  245.35  4977.3  245.98  4987.6   245.1  4994.6  241.65  4998.1  241.65
  5013.8  245.72  5023.2  245.64  5044.8  248.44  5050.2  248.93  5073.2  250.13
  5102.3   249.6  5202.2  250.91  5366.6  254.11  5451.9  257.98  5551.8  264.75
#Mann= 5 ,-1 , 0
  4595.4     .17       0  4851.1     .15       0  4905.1     .09       0
  5044.8     .15       0  5050.2     .11       0
Bank Sta=4905.1,5044.8
XS Rating Curve= 0 ,0
Exp/Cntr=0.3,0.1

Type RM Length L Ch R = 1 ,41541   ,785,785,785
BEGIN DESCRIPTION:
STEWART CREEK NORTH 83.0
END DESCRIPTION:
XS GIS Cut Line= 4
      3760327.12     10134511.41      3760575.02     10134131.87
      3760574.59      10134100.6       3760155.7     10133356.85
#Sta/Elev= 30
  4515.4  257.57  4549.6  257.34  4725.9  254.04  4754.7  254.71  4783.2  252.96
  4798.3  253.63  4921.9  252.44  4964.2  250.17  4971.6   250.7  4976.7  248.52
  4977.1  248.35 4983.54  245.25  4995.5  238.74    4999  238.74  5004.4  242.23
  5010.9  244.04  5020.3  245.24    5026  244.27  5069.4  243.93  5091.3  242.61
  5127.8   244.3  5144.6  244.05    5172  248.24  5278.3  247.86  5393.7  248.69
  5408.3  248.57  5598.2  250.84  5630.1  249.92  5673.4  251.35  5853.6   260.7
#Mann= 10 ,-1 , 0
  4515.4     .11       0  4549.6     .17       0  4976.7     .15       0
  4977.1     .17       0 4983.54     .09       0  5020.3     .17       0
  5127.8     .15       0  5278.3     .11       0  5393.7     .17       0
  5408.3     .11       0
#XS Ineff= 2 , 0
       0                    5172       0  248.24
Permanent Ineff=
       F       F
Bank Sta=4983.54,5020.3
XS Rating Curve= 0 ,0
Exp/Cntr=0.3,0.1

Type RM Length L Ch R = 1 ,40756   ,756,756,756
BEGIN DESCRIPTION:
STEWART CREEK NORTH 81.0
END DESCRIPTION:
XS GIS Cut Line= 4
      3760542.31     10134876.75      3760824.81     10134174.38
       3760941.7     10134056.73      3761262.39     10133720.56
#Sta/Elev= 30
  4077.1  263.19  4185.7  259.22  4363.5  255.32  4623.7  251.86  4723.1  248.57
  4740.7  246.19  4747.3  244.01  4752.7  245.56  4762.3  242.15  4776.9  239.26
  4794.6  243.07  4801.1  242.78  4839.9  241.51  4878.8  233.79  4895.2  236.26
  4902.3  239.03  4930.6  240.48  4965.9  239.06    5000  241.12  5008.2   244.2
  5015.4  243.08  5018.9  245.04  5022.4  246.99  5029.6  244.09  5036.5  246.24
  5043.8  246.47  5135.6  246.99    5263  250.01  5340.7  253.86  5464.6  263.36
#Mann= 5 ,-1 , 0
  4077.1     .11       0  4623.7     .17       0  4801.1     .09       0
  5008.2     .15       0  5018.9     .11       0
Bank Sta=4801.1,5008.2
XS Rating Curve= 0 ,0
Exp/Cntr=0.3,0.1

Type RM Length L Ch R = 1 ,40000   ,500,500,500
BEGIN DESCRIPTION:
STEWART CREEK NORTH 80.0
END DESCRIPTION:
XS GIS Cut Line= 3
      3760567.85     10134911.07      3761079.02     10134490.89
      3761422.68     10133795.81
#Sta/Elev= 30
  4338.3  263.22  4547.1  256.04  4583.8     255  4692.5  252.46  4808.5  249.19
  4930.7  247.83  4971.1  247.09 4981.53  242.92  4991.9  238.23    4996  233.14
  5004.7  231.88  5009.4  231.88  5012.6  235.74  5044.4  237.15  5051.9  235.91
  5057.5  238.44  5141.6  240.47    5156  242.82  5178.3  241.73  5186.5  237.37
  5192.1  240.69  5208.9  235.01  5214.5  240.12  5231.4  239.63    5237  244.11
  5370.4  244.05    5446  244.22  5585.5  249.36  5708.1  255.48  5775.4  261.49
#Mann= 10 ,-1 , 0
  4338.3     .11       0  4547.1     .17       0  4583.8     .11       0
  4692.5     .17       0  4808.5     .11       0  4930.7     .17       0
 4981.53     .09       0    5156     .15       0  5370.4     .17       0
  5585.5     .11       0
#XS Ineff= 2 , 0
       0                  5245.2       0  244.24
Permanent Ineff=
       F       F
Bank Sta=4981.53,5156
XS Rating Curve= 0 ,0
Exp/Cntr=0.3,0.1

Type RM Length L Ch R = 1 ,39500   ,500,500,500
BEGIN DESCRIPTION:
STEWART CREEK NORTH 79.0
END DESCRIPTION:
XS GIS Cut Line= 3
      3761481.66     10135058.88      3761493.15     10134451.89
      3761617.85     10133961.08
#Sta/Elev= 30
  4392.9  248.44  4400.7  247.62  4472.1  247.03  4620.7  246.63  4766.8  245.14
  4840.8  242.61  4850.8  241.04  4865.1  236.77  4870.8  234.45  4890.8  236.11
  4910.8  239.13  4930.8  241.05  4940.8  241.12  4960.8   235.1  4970.8  234.09
    4980  231.51    4985  233.45  4990.8   231.8  4995.5  228.08    5003  228.58
  5011.2  233.29  5038.2  241.59  5062.7  242.36  5125.2  241.31    5135  242.29
  5176.2  241.06  5207.2   242.5  5318.3  245.06  5413.6  248.15  5506.4  254.25
#Mann= 7 ,-1 , 0
  4392.9     .17       0  4472.1     .11       0  4766.8     .17       0
  4865.1     .15       0  4940.8     .09       0  5038.2     .15       0
  5318.3     .11       0
Bank Sta=4940.8,5038.2
XS Rating Curve= 0 ,0
Exp/Cntr=0.3,0.1

Type RM Length L Ch R = 1 ,39000   ,500,500,500
BEGIN DESCRIPTION:
STEWART CREEK NORTH 78.0
END DESCRIPTION:
XS GIS Cut Line= 3
      3761581.47     10135163.04      3761931.56     10134375.67
      3761872.28     10133947.75
#Sta/Elev= 30
  4138.3  252.41  4151.4  252.73  4190.3  250.14    4219  249.66  4260.1   246.4
  4265.5  247.04  4294.3  244.19    4312  245.45  4358.5     244  4468.8  244.19
    4543  241.53  4688.2  240.63  4698.6  241.36    4819  239.36  4860.3  239.88
  4895.6  240.56  4926.1  239.99  4939.4  239.88  4961.3  236.37  4972.2  236.14
  4978.1  234.51  4983.6  235.02  4997.3  227.58  5004.8  228.08  5014.7  232.87
    5045  238.42  5075.3  240.12  5202.5  241.41  5337.8   246.6    5432  253.57
#Mann= 6 ,-1 , 0
  4138.3     .11       0    4543     .17       0  4860.3     .15       0
  4926.1     .09       0  5075.3     .15       0  5202.5     .11       0
Bank Sta=4926.1,5075.3
XS Rating Curve= 0 ,0
Exp/Cntr=0.3,0.1

Type RM Length L Ch R = 1 ,38500   ,500,500,500
BEGIN DESCRIPTION:
STEWART CREEK NORTH 77.0
END DESCRIPTION:
XS GIS Cut Line= 3
      3762145.72     10135045.83      3762321.99     10134396.01
      3762089.71     10133905.21
#Sta/Elev= 30
  4326.7  246.63  4487.1  243.51  4509.8  243.98  4544.5  242.53  4624.1  241.71
  4642.5     240  4658.8  240.88  4670.7  240.38  4771.5  237.58  4847.5  238.37
  4906.8     237  4906.9     237  4953.3  237.43  4961.8   235.3    4967  235.52
  4984.4  230.71  4992.3   225.3  4997.3   225.3    5000  228.63  5005.5  228.63
  5016.2  233.96  5021.7  232.42  5027.6   236.9  5293.1  242.12  5381.6  242.72
  5396.8  241.27  5403.8  241.35  5450.5     245  5481.2  245.46    5543  248.21
#Mann= 8 ,-1 , 0
  4326.7     .11       0  4670.7     .17       0  4771.5     .15       0
  4906.8     .17       0  4906.9     .15       0  4953.3     .09       0
  5027.6     .15       0  5450.5     .11       0
#XS Ineff= 2 , 0
       0  4673.6  240.44               0
Permanent Ineff=
       F       F
Bank Sta=4953.3,5027.6
XS Rating Curve= 0 ,0
Exp/Cntr=0.3,0.1

Type RM Length L Ch R = 1 ,38000   ,500,500,500
BEGIN DESCRIPTION:
STEWART CREEK NORTH 76.0
END DESCRIPTION:
XS GIS Cut Line= 3
      3762577.42     10135183.36      3762737.89     10134588.46
      3762788.08     10133821.87
#Sta/Elev= 30
       0  244.49   126.7  243.28     179   241.6   240.6  241.22   288.4  239.79
   344.2  238.77   437.4   239.9   448.1  238.64   458.1  239.64   482.8  238.37
   509.9  239.76   582.4  236.62   592.2  234.43   597.4  234.36   603.1   228.9
   612.2  225.82   623.6  226.32   633.6  231.15   643.6  233.92   653.6  235.57
   773.9  235.67   783.9  234.89   793.9  232.84     814  231.92   842.1  235.05
   884.1  234.51   914.2  235.93   993.8  236.43    1275   241.7  1384.4  244.51
#Mann= 5 ,-1 , 0
       0     .11       0   288.4     .17       0   582.4     .09       0
   653.6     .17       0   793.9     .11       0
Bank Sta=582.4,653.6
XS Rating Curve= 0 ,0
Exp/Cntr=0.3,0.1

Type RM Length L Ch R = 1 ,37500   ,500,500,500
BEGIN DESCRIPTION:
STEWART CREEK NORTH 75.0
END DESCRIPTION:
XS GIS Cut Line= 3
      3762945.47     10135200.72       3763075.9     10134679.97
      3763467.85     10134161.07
#Sta/Elev= 30
       0  242.97    61.5  243.36    82.1  241.32   110.3  240.63   185.2  239.79
   205.8  240.47     239  239.25   370.8  236.82     412  234.42   422.3  233.41
   432.6  230.94     445  232.21   453.2  233.99   463.5  234.36   494.5  234.89
   504.8  233.21   515.1  231.37   522.3  228.72   527.4  225.28   533.7  222.56
     545   223.3   559.6  232.12   573.1  234.09   601.3   234.4   651.2  234.45
   865.6  235.86   930.1  237.38   994.6  239.72  1123.6  247.84  1187.1   252.7
#Mann= 6 ,-1 , 0
       0     .11       0     239     .17       0   504.8     .09       0
   559.6     .15       0   601.3     .17       0   651.2     .11       0
Bank Sta=504.8,559.6
XS Rating Curve= 0 ,0
Exp/Cntr=0.3,0.1

Type RM Length L Ch R = 1 ,37000   ,500,500,500
BEGIN DESCRIPTION:
STEWART CREEK NORTH 74.0
END DESCRIPTION:
XS GIS Cut Line= 3
      3763139.63     10135163.03       3763420.9     10134901.17
       3763725.6     10134347.01
#Sta/Elev= 30
  4615.7  241.68  4686.5  242.11    4708  240.07  4806.7  238.31  4842.4  235.75
  4849.2  237.07  4877.5  237.71  4927.4  235.98  4955.2  231.35  4962.6  228.51
  4969.4  227.45  4983.6  227.01  4990.9  224.92  4996.4  220.53  5001.7     220
  5008.1     220  5011.5  222.61    5021  227.79  5034.9  230.91  5057.2   233.5
  5108.2  230.79  5124.3  232.95  5200.7  232.95  5217.1  233.38  5276.8  231.85
  5308.2  232.89  5410.9  237.85  5445.4  240.29  5483.3  241.55  5632.4   251.4
#Mann= 4 ,-1 , 0
  4615.7     .11       0  4955.2     .07       0  5034.9     .15       0
  5200.7     .11       0
Bank Sta=4955.2,5034.9
XS Rating Curve= 0 ,0
Exp/Cntr=0.3,0.1

Type RM Length L Ch R = 1 ,36500   ,484,484,484
BEGIN DESCRIPTION:
STEWART CREEK NORTH 73.0
END DESCRIPTION:
XS GIS Cut Line= 4
      3763157.04     10135310.58      3763647.45     10135163.02
      3763859.31     10134962.12       3764129.2     10134733.35
#Sta/Elev= 30
  4195.9  243.16  4491.8  238.75  4541.4  236.05  4723.7  231.97  4780.3  232.55
  4858.4  231.18  4865.3  232.05  4893.6  230.78  4929.1  232.06  4950.2  228.94
  4964.4  227.81  4971.3  225.17  4978.5  224.32  4992.7  218.63  4993.8  217.27
    5007  218.81  5013.6  224.17  5021.3  225.87  5027.8   229.1  5056.4  232.39
  5088.6  234.36  5113.6  236.91  5120.1  238.93  5148.7  238.28    5163  240.79
  5177.3  241.24  5183.8  239.37  5255.3  240.58  5261.8  243.27  5353.8  249.15
#Mann= 4 ,-1 , 0
  4195.9     .11       0  4950.2     .09       0  5027.8     .15       0
  5088.6     .17       0
Bank Sta=4950.2,5027.8
XS Rating Curve= 0 ,0
Exp/Cntr=0.3,0.1

Type RM Length L Ch R = 1 ,36016   ,158,158,158
BEGIN DESCRIPTION:
STEWART CREEK NORTH 72.0
END DESCRIPTION:
XS GIS Cut Line= 3
      3763050.48     10135454.01      3764010.26     10135347.28
      3765052.29     10135143.34
#Sta/Elev= 30
  4034.3  245.91  4202.7  244.86  4463.7  238.18  4468.7  240.02  4553.9  236.31
  4735.2  231.49  4740.3  233.41  4830.8  228.84  4916.3  230.63  4921.3  228.14
  4937.2  228.22  5006.2   216.5  5012.9   216.5  5048.5  228.11    5056  230.78
  5107.5  232.64  5112.6  230.08    5256  230.72    5454   234.9  5627.6  233.78
  5632.7  235.97  5730.7  238.74  5735.7  240.83  5838.8  241.91  5895.4  245.94
  5941.8  244.85  5946.9  247.45  5993.3  246.77  5998.4  249.08  6061.8  250.35
#Mann= 6 ,-1 , 0
  4034.3     .11       0  4553.9    .125       0  4937.2     .09       0
  5048.5    .125       0    5256     .11       0    5454    .125       0
Bank Sta=4937.2,5048.5
XS Rating Curve= 0 ,0
Exp/Cntr=0.3,0.1

Type RM Length L Ch R = 1 ,35858   ,758,758,758
BEGIN DESCRIPTION:
STEWART CREEK NORTH 71.0
END DESCRIPTION:
XS GIS Cut Line= 3
      3763097.85     10135653.32      3764041.18      10135501.9
      3765130.69     10135337.84
#Sta/Elev= 30
  4044.6  248.65  4358.6  240.93  4781.6  236.92  4786.7  235.04  4843.6  234.81
  4895.4  230.41  4925.7  225.92    4946  225.31  4972.5  219.44  4986.5  219.17
  4992.3  216.78  5006.7  217.36  5035.6  225.78  5057.3   229.1  5173.5  230.31
  5370.3  228.11  5421.4  225.28    5482  229.01  5502.3  234.13  5513.3  234.68
  5562.9  234.61  5577.3   233.7  5583.2  231.24  5593.3  229.86  5805.7  234.93
  5906.8  239.52  5987.7  241.21    6018  239.85  6068.6  243.03  6101.8  243.25
#Mann= 3 , 0 , 0
  4044.6     .11       0  4925.7     .06       0  5035.6     .11       0
#XS Ineff= 2 , 0
       0                  5067.4       0  229.35
Permanent Ineff=
       F       F
Bank Sta=4925.7,5035.6
XS Rating Curve= 0 ,0
Exp/Cntr=0.3,0.1

Type RM Length L Ch R = 1 ,35100   ,600,600,600
BEGIN DESCRIPTION:
STEWART CREEK NORTH 70.0
END DESCRIPTION:
XS GIS Cut Line= 3
      3764066.28     10136307.67      3764622.29     10135890.03
       3765171.2     10135372.95
#Sta/Elev= 30
  4304.6  242.54    4510  241.83  4645.4  238.73  4839.1  230.27  4903.7  225.13
  4909.9   223.5  4939.1   222.4  4953.7  222.54  4959.9  224.53  4974.5  221.55
  4991.5  213.06  5024.3  214.09  5045.8  217.82  5052.6     221  5059.9  219.03
  5066.8  222.84  5080.9  224.57  5102.4  229.18  5144.9  231.31  5201.1  224.08
  5208.4   225.6  5279.2  227.37  5335.8  226.72  5356.9  228.19  5462.9  228.77
  5505.4  231.84  5526.8  230.86  5661.1  236.18  5696.3   240.1  5754.1  242.83
#Mann= 3 , 0 , 0
  4304.6     .11       0  4903.7     .06       0  5080.9     .11       0
#XS Ineff= 2 , 0
       0                  5144.9       0  231.31
Permanent Ineff=
       F       F
Bank Sta=4903.7,5080.9
XS Rating Curve= 0 ,0
Exp/Cntr=0.3,0.1

Type RM Length L Ch R = 1 ,34500   ,500,500,500
BEGIN DESCRIPTION:
STEWART CREEK NORTH 69.0
END DESCRIPTION:
XS GIS Cut Line= 3
      3764823.28     10136773.62      3765032.05     10136129.72
      3765419.39      10135590.4
#Sta/Elev= 30
  4323.1  235.02  4353.1  235.62  4367.8  233.92  4399.4  233.85    4473  236.22
    4536  236.53  4599.1   231.8  4715.4  226.91  4788.3  224.69  4907.3  223.34
  4914.5  220.53    4934  217.63  4939.2  215.81    4946  218.63    4966  221.22
  4971.2  215.35  4977.6  215.42  4999.2  211.22  5017.7  211.97  5023.8  217.87
  5032.4  218.14  5038.5  223.15  5053.3  224.85  5311.1  223.82  5382.3  225.96
  5441.2  225.86  5518.6  229.21    5577   234.7  5589.8  237.16    5664  239.28
#Mann= 3 , 0 , 0
  4323.1     .11       0  4907.3     .06       0  5038.5     .11       0
Bank Sta=4907.3,5038.5
XS Rating Curve= 0 ,0
Exp/Cntr=0.3,0.1

Type RM Length L Ch R = 1 ,34000   ,500,500,500
BEGIN DESCRIPTION:
STEWART CREEK NORTH 68.0
END DESCRIPTION:
XS GIS Cut Line= 4
      3764856.22     10136794.61      3765358.02     10136244.73
      3765378.61     10136126.64      3765467.85      10135611.1
#Sta/Elev= 30
  4135.7  235.74  4146.4  234.32  4167.6  233.22    4189  233.85  4238.3  232.21
    4366  231.85  4507.2  225.29  4592.3  222.64    4670  221.98  4797.7  223.39
  4934.6  222.41  4954.9  223.04  4968.3  221.89  4985.3   218.6  4995.2  212.83
    5000  212.83  5001.9  209.06  5009.4  209.06  5015.8  216.62  5022.9  221.44
  5027.9  220.86  5036.1  222.91  5046.2  223.29  5066.5  222.52    5097  223.32
  5188.3  222.97  5330.4  226.29  5411.6  230.89  5490.8  237.47  5523.2  238.76
#Mann= 3 , 0 , 0
  4135.7     .11       0  4968.3     .06       0  5022.9     .11       0
Bank Sta=4968.3,5022.9
XS Rating Curve= 0 ,0
Exp/Cntr=0.3,0.1

Type RM Length L Ch R = 1 ,33500   ,500,500,500
BEGIN DESCRIPTION:
STEWART CREEK NORTH 67.0
END DESCRIPTION:
XS GIS Cut Line= 3
      3764904.13     10136839.55      3765730.73     10136284.98
      3766254.03     10136120.96
#Sta/Elev= 30
  4004.6  232.76    4100  229.85  4553.2  221.45  4892.3  221.95  4900.2  219.87
  4907.3  216.07  4913.3  218.51  4922.2  215.12  4928.3  216.73  4943.3  214.58
  4949.3     217  4958.3  215.17  4964.3  217.66  4979.3   212.6  4985.3  214.37
  5003.7  208.15  5017.9  209.91  5026.5  208.82  5031.7  210.63  5049.4  209.97
  5058.9  214.94  5064.2  215.24  5070.3  217.94  5096.6  221.96    5264   227.2
  5501.6   238.8  5510.5  237.42    5521  237.86  5528.8   239.8  5548.4  240.18
#Mann= 3 , 0 , 0
  4004.6     .06       0  4892.3     .07       0  5096.6     .15       0
#XS Ineff= 2 , 0
       0                    5129       0  222.82
Permanent Ineff=
       F       F
Bank Sta=4892.3,5096.6
XS Rating Curve= 0 ,0
Exp/Cntr=0.3,0.1

Type RM Length L Ch R = 1 ,33000   ,500,500,500
BEGIN DESCRIPTION:
STEWART CREEK NORTH 66.0
END DESCRIPTION:
XS GIS Cut Line= 3
      3765341.51     10137112.11      3765847.24     10136640.81
      3766267.84     10136161.08
#Sta/Elev= 30
  4308.7  231.49  4363.4  227.78  4497.7  222.56  4639.4  220.45  4830.5  218.98
  4915.5  220.93  4936.5  220.18  4972.1  216.97    4979  217.56  4993.1  211.84
    4997  207.67    5000  207.67  5002.6  206.53  5012.3  206.53  5014.1  209.26
  5021.6  210.83  5028.3  217.04  5035.9  218.31  5042.5  220.57    5163  219.24
  5297.8  222.44  5318.8  224.06  5397.4  226.49    5518   234.4  5567.3  234.77
    5574  237.22  5588.2  237.97  5624.2  238.79  5630.9  237.39    5638  237.49
#Mann= 3 , 0 , 0
  4308.7     .11       0  4936.5     .06       0  5042.5     .11       0
Bank Sta=4936.5,5042.5
XS Rating Curve= 0 ,0
Exp/Cntr=0.3,0.1

Type RM Length L Ch R = 1 ,32500   ,500,500,500
BEGIN DESCRIPTION:
STEWART CREEK NORTH 65.0
END DESCRIPTION:
XS GIS Cut Line= 3
      3765667.86     10137461.06      3766018.33     10137052.09
      3766737.41     10136300.33
#Sta/Elev= 30
  4461.4  235.81  4759.4  222.05  4843.9  216.32  4908.7  218.26  4915.2  216.56
  4943.8  216.06  4950.4  213.47    4958  214.44  4964.6  212.02  4972.3  214.61
  4978.9  210.23  4986.6  212.02  4992.5  205.69  5002.2  205.69  5007.4  209.57
  5014.7   208.8  5021.6   211.4  5028.8  210.94  5035.7  214.76    5064  218.37
  5078.2  219.85  5177.3  219.85  5389.2  217.31  5438.9  220.12  5481.4   218.3
  5792.4  227.06  5863.2  231.21  5919.8  232.23  6004.7  239.71  6040.3  239.57
#Mann= 3 , 0 , 0
  4461.4     .11       0  4908.7     .06       0    5064     .11       0
Bank Sta=4908.7,5064
XS Rating Curve= 0 ,0
Exp/Cntr=0.3,0.1

Type RM Length L Ch R = 1 ,32000   ,500,500,500
BEGIN DESCRIPTION:
STEWART CREEK NORTH 64.0
END DESCRIPTION:
XS GIS Cut Line= 3
      3766048.46     10137642.28      3766298.97     10137266.41
       3766947.1      10136650.8
#Sta/Elev= 30
  4548.3  233.68  4793.4  222.11  4829.4  221.23  4874.2  218.14  4916.6  218.93
  4937.6  217.75  4958.6  217.98  4967.7  216.22  4973.7     217  4982.4  214.78
  4988.7   211.2    5000  211.04  5002.9   205.9  5005.3  205.39  5015.1  205.39
  5017.1   206.9  5031.2   211.3  5045.4  212.17  5052.7  216.76  5059.6   216.4
  5066.8   218.2  5116.2   217.1  5201.1  218.66  5377.9  216.19  5618.5  219.02
  5667.9  221.52  5703.1  224.97  5781.2   238.2  5809.5  239.62  5893.9   240.4
#Mann= 3 , 0 , 0
  4548.3     .11       0  4973.7     .06       0  5052.7     .11       0
Bank Sta=4973.7,5052.7
XS Rating Curve= 0 ,0
Exp/Cntr=0.3,0.1

Type RM Length L Ch R = 1 ,31500   ,299,299,299
BEGIN DESCRIPTION:
STEWART CREEK NORTH 63.0
END DESCRIPTION:
XS GIS Cut Line= 4
      3766222.15     10137753.17      3766667.98     10137382.69
      3766690.83     10137340.33      3767087.86      10136791.6
#Sta/Elev= 30
  4372.2   233.9  4526.6  229.69  4740.2   218.7    4761  219.86  4846.9  211.43
  4860.7  215.45  4896.4  216.12  4910.7  215.65  4917.2  211.93  4925.1   214.8
  4931.6  209.97  4945.9  214.22  4955.6  211.63  4960.8  206.52  4966.4  211.52
  4982.7  204.86  4988.3  207.31  4996.7   204.3  5004.4  205.78  5006.4   203.4
  5016.4   203.4  5019.1  210.25  5025.2  210.06  5033.8  215.04  5039.9  212.93
  5048.5  216.61    5398  215.84  5433.6  219.06  5548.8   238.5  5677.3  240.29
#Mann= 3 , 0 , 0
  4372.2     .11       0  4896.4     .06       0  5048.5     .11       0
Bank Sta=4896.4,5048.5
XS Rating Curve= 0 ,0
Exp/Cntr=0.3,0.1

Type RM Length L Ch R = 1 ,31201   ,200,200,200
BEGIN DESCRIPTION:
Mapping XS 4e96840b
END DESCRIPTION:
XS GIS Cut Line= 3
      3766521.52     10137939.56      3766965.74     10137337.71
      3767199.78     10136910.22
#Sta/Elev= 30
  4252.1  230.27  4334.8  227.09  4541.5  222.59  4721.1  213.95  4834.4  215.93
  4948.6  215.74  4984.1  212.12  4992.5  209.12  4997.7  203.54  5002.6  202.64
  5012.7  202.64  5013.2  203.14  5014.2   209.4  5030.3  215.75  5079.6  216.24
  5133.1  211.99  5155.5  214.67    5183  213.45  5199.1  215.36  5226.6  214.59
  5270.2  219.75  5351.8  224.98  5389.7  228.95  5411.5  228.67  5427.6  231.13
  5433.3  230.31  5449.4  232.94  5455.1  232.24  5471.2   234.9  5487.5  235.43
#Mann= 3 , 0 , 0
  4252.1     .11       0  4948.6     .06       0  5030.3     .11       0
Bank Sta=4948.6,5030.3
XS Rating Curve= 0 ,0
Exp/Cntr=0.3,0.1

Type RM Length L Ch R = 1 ,31001   ,213,213,213
BEGIN DESCRIPTION:
STEWART CREEK NORTH 62.0
END DESCRIPTION:
XS GIS Cut Line= 3
      3766614.57     10138010.77      3767141.15     10137360.68
      3767362.88     10136920.14
#Sta/Elev= 30
  4163.4  231.21  4371.3  226.64  4591.9  215.94  4620.6  216.53  4742.1  213.39
    4806  214.87  4911.6  213.86  4933.9  215.47  4969.1  215.16  4975.6  213.43
  4999.4  202.71  5009.5  202.71    5010  203.21  5010.8  208.31  5026.8  213.24
  5033.2  213.58  5049.1  209.06  5071.4  210.57  5077.9  213.55  5088.1  214.16
  5138.4  213.71  5155.1  214.92    5183  220.49    5222  214.77  5272.3   216.6
  5316.9  226.58  5339.2  225.92  5383.9  231.26  5458.6  234.84  5493.2  239.04
#Mann= 3 , 0 , 0
  4163.4     .11       0  4969.1     .06       0  5155.1     .11       0
#XS Ineff= 2 , 0
       0  4620.6  216.53    5183       0  220.49
Permanent Ineff=
       F       F
Bank Sta=4969.1,5155.1
XS Rating Curve= 0 ,0
Exp/Cntr=0.3,0.1

Type RM Length L Ch R = 1 ,30788   ,307,307,307
BEGIN DESCRIPTION:
Mapping XS 63247e3c
END DESCRIPTION:
XS GIS Cut Line= 3
      3766734.07      10138075.7      3767331.93     10137413.31
      3767550.86     10137051.14
#Sta/Elev= 30
  4107.7  230.13  4234.3  227.76  4347.2  224.22  4666.2   212.4  4687.2   213.1
  4750.7  212.22  4786.6   213.8  4906.9  213.33  4956.2  214.57  4977.2  213.63
  4998.1  208.59  5000.1  204.46  5010.2  204.46  5014.3  208.54  5020.6  212.84
  5026.5  214.53  5078.8  212.74  5094.3   214.4  5121.5  213.85  5158.4  219.84
  5166.2  219.19  5179.7  216.33  5195.3  215.49  5216.6  220.02    5238  220.89
  5253.5  223.93    5269  229.13  5283.1  231.47    5364  233.19  5423.2  232.94
#Mann= 3 ,-1 , 0
  4107.7     .11       0  4956.2     .06       0  5026.5     .11       0
#XS Ineff= 2 , 0
       0                  5158.4       0  219.84
Permanent Ineff=
       F       F
Bank Sta=4956.2,5026.5
XS Rating Curve= 0 ,0
Exp/Cntr=0.3,0.1

Type RM Length L Ch R = 1 ,30481   ,481,481,481
BEGIN DESCRIPTION:
STEWART CREEK NORTH 61.0
END DESCRIPTION:
XS GIS Cut Line= 3
      3766851.25     10138127.57      3767468.52     10137605.73
      3767722.14     10137104.65
#Sta/Elev= 30
  4191.7  229.04  4435.7  223.37  4754.3  212.39  4868.2  210.98    4974  213.25
    4991  203.49  5004.8  204.02  5016.4  207.13  5026.9  206.51  5032.5  211.01
  5049.2  207.35  5054.8   211.6  5093.7  208.65  5099.3  212.35  5106.1  210.09
    5116  210.57  5121.6  213.91  5150.9  214.01  5160.6  212.18  5166.2  214.09
  5188.4  213.99  5205.1  211.74  5227.4  215.19  5249.7  213.62  5285.4  220.16
  5322.1  215.74  5344.4  220.09  5366.7  221.78  5405.6   231.9  5561.6  232.67
#Mann= 3 ,-1 , 0
  4191.7     .11       0    4974     .06       0  5121.6     .11       0
#XS Ineff= 3 ,-1
  4967.4  4676.2  213.81  5128.5  5227.4   214.2  5227.4  5285.4  215.19
Permanent Ineff=
       F       F       F
Bank Sta=4974,5121.6
XS Rating Curve= 0 ,0
Exp/Cntr=0.3,0.1

Type RM Length L Ch R = 1 ,30000   ,500,500,500
BEGIN DESCRIPTION:
STEWART CREEK NORTH 60.0
END DESCRIPTION:
XS GIS Cut Line= 3
      3767015.96     10138409.18      3767854.73     10137807.94
      3767842.74     10137125.04
#Sta/Elev= 30
    3968  228.29  4132.1  223.54  4357.1  220.36  4563.5  212.18  4792.9  210.71
  4813.8  207.59  4819.9  202.14  4843.2  201.03  4849.4   203.5  4864.1   204.7
  4870.3  208.08    4885  210.21  4920.6  212.27  4964.8  212.35  4979.2  207.93
  4985.7  207.91  4991.9  200.89  4993.8   200.1  5003.9   200.1  5016.9  209.18
  5026.9  212.05  5046.9  214.88  5076.9  211.38  5236.9  212.22  5336.9  215.06
  5356.9  213.56  5416.9  226.64  5446.9  228.86    5557  232.48    5683  232.33
#Mann= 5 ,-1 , 0
    3968     .11       0  4357.1    .125       0  4563.5     .11       0
  4964.8     .06       0  5026.9     .11       0
#XS Ineff= 3 ,-1
  4964.8  4677.4  212.35  4677.4  4548.6  212.45  5046.9  5376.9  214.88
Permanent Ineff=
       F       F       F
Bank Sta=4964.8,5026.9
XS Rating Curve= 0 ,0
Exp/Cntr=0.3,0.1

Type RM Length L Ch R = 1 ,29500   ,500,500,500
BEGIN DESCRIPTION:
STEWART CREEK NORTH 59.0
END DESCRIPTION:
XS GIS Cut Line= 4
      3767717.87     10138861.05      3768269.19     10137907.34
      3768287.71     10137881.88      3768517.84     10137411.09
#Sta/Elev= 30
  3898.4  228.06  4249.4  213.41  4741.6  209.87  4784.8  201.68  4806.2  199.66
  4806.7  199.16  4817.9  199.66  4849.4   200.6  4902.5  209.89  4945.5  210.87
  4951.3  209.21  4967.1  209.63  4972.9  205.32  4982.8  206.98  4988.6  201.11
    5000  200.47  5010.1  202.44  5018.6  201.89  5028.9  208.55  5046.1  211.36
  5085.6  210.49  5198.2  213.34  5210.5  215.23  5248.8  215.35  5299.5  221.37
  5338.8  217.23  5389.4  217.27    5422  220.13  5496.5  232.81  5555.5  237.38
#Mann= 5 ,-1 , 0
  3898.4     .11       0  4806.2     .09       0  4817.9     .11       0
  4945.5     .07       0  5046.1     .11       0
#XS Ineff= 2 ,-1
                          4945.5  4592.4  210.87
Permanent Ineff=
       F       F
Bank Sta=4945.5,5046.1
XS Rating Curve= 0 ,0
Exp/Cntr=0.3,0.1

Type RM Length L Ch R = 1 ,29000   ,500,500,500
BEGIN DESCRIPTION:
STEWART CREEK NORTH 58.0
END DESCRIPTION:
XS GIS Cut Line= 4
       3767857.7     10138906.42      3768621.04     10138092.82
      3768631.31     10138071.16      3768756.35      10137399.7
#Sta/Elev= 30
  3860.4  228.91  4281.6  212.54  4699.2  209.61  4762.7   207.6    4770  204.42
  4776.8   205.8  4784.1  202.58    4791  203.73  4798.3  201.08  4812.5  200.68
  4882.8  200.38  4925.3  204.96  4932.6  207.61  4953.7  207.96  4967.8  207.74
  4973.8   204.7  4981.9  205.77    4989  201.83  5002.6   202.1  5006.5   199.7
  5017.2   199.7  5030.6   208.2    5078  210.24  5285.8  210.16  5338.5  212.28
  5417.1  221.41    5468   217.9  5539.2  218.06  5607.3     232    5683  236.58
#Mann= 5 ,-1 , 0
  3860.4     .11       0  4699.2     .15       0  4953.7     .09       0
  5030.6     .15       0    5078     .11       0
#XS Ineff= 2 , 0
       0    4579  211.32  5071.3       0  210.57
Permanent Ineff=
       F       F
Bank Sta=4953.7,5030.6
XS Rating Curve= 0 ,0
Exp/Cntr=0.3,0.1

Type RM Length L Ch R = 1 ,28500   ,500,500,500
BEGIN DESCRIPTION:
STEWART CREEK NORTH 57.0
END DESCRIPTION:
XS GIS Cut Line= 4
      3769067.88     10138867.43      3769043.78     10137869.73
      3769032.95     10137827.08      3768967.85     10137311.07
#Sta/Elev= 30
    3958  223.14  4024.4  222.43  4264.5  216.45  4324.5  216.12  4444.5   213.8
  4614.6  208.92  4694.6  207.99  4834.6  209.29  4864.6  208.78  4884.6  207.88
  4894.6  203.75  4899.2  200.48  4910.5  200.98  5116.9     201  5156.4  203.16
  5161.4  207.32  5197.6  205.39  5241.7  207.04    5248  205.61  5268.1  205.52
  5298.4  208.36  5316.9  210.48    5322     212  5338.7  214.94  5348.8  218.06
  5358.8   219.4  5368.9  218.38  5409.2  223.26  5449.1  226.68  5520.1  234.05
#Mann= 4 ,-1 , 0
    3958     .11       0  4864.6     .09       0  5298.4     .15       0
  5449.1     .11       0
Bank Sta=4864.6,5298.4
XS Rating Curve= 0 ,0
Exp/Cntr=0.3,0.1

Type RM Length L Ch R = 1 ,28000   ,500,500,500
BEGIN DESCRIPTION:
STEWART CREEK NORTH 56.0
END DESCRIPTION:
XS GIS Cut Line= 3
      3769867.87     10138511.09      3769372.55     10137723.97
      3769047.72     10137254.61
#Sta/Elev= 30
    4070  220.81  4164.5  218.95  4214.3  217.37  4229.6  216.07  4256.5  216.39
  4371.5  211.99  4483.6  208.09  4752.4  206.76  4779.5   205.4    4838  207.32
  4919.6  208.07  4925.5  208.94  4932.5  208.61  4940.8  206.62  4946.7  206.76
  4956.1  203.58  4971.8   200.5  5027.8     201  5055.2  203.13    5064  206.67
  5070.1  206.69    5085  209.96  5120.8  211.72  5149.5  211.43  5239.6  213.03
  5320.8  215.52  5401.2  216.68  5487.7  224.01  5529.6  231.05  5570.8  234.47
#Mann= 6 ,-1 , 0
    4070     .15       0  4256.5     .17       0  4371.5     .11       0
  4946.7     .07       0    5064     .11       0  5239.6     .11       0
Bank Sta=4946.7,5064
XS Rating Curve= 0 ,0
Exp/Cntr=0.3,0.1

Type RM Length L Ch R = 1 ,27500   ,500,500,500
BEGIN DESCRIPTION:
STEWART CREEK NORTH 55.0
END DESCRIPTION:
XS GIS Cut Line= 3
      3769917.85     10138411.06      3769861.58     10137748.74
      3769789.82     10137190.74
#Sta/Elev= 30
  4335.3  217.76  4397.4  217.01  4431.1  215.55  4586.2  209.78  4694.3  206.81
  4765.3  206.81  4790.1  207.14  4897.3  209.31  4907.3  209.16  4917.4  207.09
 4920.23  205.75  4931.9   200.5  4943.4     201  5048.1     201  5065.8  205.55
  5070.9  205.74  5078.3  209.09  5088.4  210.14    5159  210.36  5189.2  207.31
  5219.5  206.89  5224.9  207.52  5229.9  207.07  5259.8   210.5  5269.9  210.97
  5370.7  212.73  5435.5  212.49  5458.4  211.65  5501.8  212.68  5562.6  217.95
#Mann= 8 ,-1 , 0
  4335.3     .15       0  4431.1     .11       0  4694.3     .15       0
  4765.3     .11       0  4790.1     .15       0 4920.23     .07       0
  5070.9     .15       0  5435.5     .11       0
#XS Ineff= 2 , 0
       0  4897.3  209.31  5128.7       0  210.58
Permanent Ineff=
       F       F
Bank Sta=4920.23,5070.9
XS Rating Curve= 0 ,0
Exp/Cntr=0.3,0.1

Type RM Length L Ch R = 1 ,27000   ,410,410,410
BEGIN DESCRIPTION:
STEWART CREEK NORTH 54.0
END DESCRIPTION:
XS GIS Cut Line= 3
      3770546.74     10138308.72      3770350.81     10137841.44
      3770171.76     10137121.26
#Sta/Elev= 30
  4493.3  215.55    4532  215.63  4566.7  215.95  4711.6  214.43  4812.2  209.47
  4881.1  208.62  4888.9  207.33  4894.3  207.89  4902.5  205.54  4924.5  202.82
  4929.8   200.5  4941.4     201    5021     201  5029.6  202.66  5034.7  202.23
  5070.9  202.76    5076     201  5248.5     201  5577.4     201  5587.7   201.6
    5598  203.16  5608.2  205.81  5613.4  204.31  5618.6  207.65  5628.9  209.94
  5654.7  210.82  5701.2  214.87    5732  219.73  5739.8  222.19  5742.1  222.19
#Mann= 6 ,-1 , 0
  4493.3     .17       0    4532     .11       0  4902.5     .15       0
  4924.5     .06       0  5029.6     .11       0  5248.5     .11       0
Bank Sta=4924.5,5029.6
XS Rating Curve= 0 ,0
Exp/Cntr=0.3,0.1

Type RM Length L Ch R = 1 ,26590   ,124,124,124
BEGIN DESCRIPTION:
STEWART CREEK NORTH 53.0
END DESCRIPTION:
XS GIS Cut Line= 3
      3770906.67      10138262.2      3770713.71     10137689.54
      3770500.53     10137118.32
#Sta/Elev= 30
  4395.7  212.28  4499.4  209.97  4554.6  207.71  4574.5  206.95  4679.6  204.95
  4745.1  203.27  4811.4  203.64  4889.8   204.3  4934.9  204.24  4940.2  202.02
  4956.2  202.64  4966.1   200.5  5051.7     201  5084.5 205.094  5259.9  206.24
  5297.2  205.86  5315.1   203.8  5320.5  207.18  5345.5  204.69  5350.8  207.89
  5370.4  206.24  5377.3  208.77  5385.2  208.48  5400.7   207.4  5406.1  208.77
  5431.1  208.15  5478.7  209.61  5532.1  209.73  5593.6  212.23  5609.7  212.71
#Mann= 11 ,-1 , 0
  4395.7     .15       0  4554.6     .11       0  4574.5     .15       0
  4679.6     .11       0  4811.4     .15       0  4889.8     .11       0
  4934.9     .06       0  5084.5     .11       0  5377.3     .11       0
  5385.2    .125       0  5593.6     .15       0
Bank Sta=4934.9,5084.5
XS Rating Curve= 0 ,0
Exp/Cntr=0.3,0.1

Type RM Length L Ch R = 1 ,26466   ,466,466,466
BEGIN DESCRIPTION:
Mapping XS 991fa303
END DESCRIPTION:
XS GIS Cut Line= 5
      3771087.33     10138103.78      3770809.39     10137617.39
       3770708.8     10137310.11      3770690.24      10137110.1
      3770705.89     10136964.61
#Sta/Elev= 30
       0  213.52    83.7  211.26   154.4   205.5   207.6  203.34   229.2  202.87
     245  204.66   272.4  205.16   347.3  203.88   383.2  203.87   412.1  205.69
   440.8  205.32   449.5  201.41   455.3  203.06   463.8     201   514.3  200.48
   598.4     201   608.5  202.84     630  204.15   703.6  203.49   883.5  205.05
   942.8  207.93   962.9  207.45  1013.1  207.16  1023.2  207.45  1033.2  209.47
  1108.7  211.32  1123.7  209.79  1173.9  210.24  1200.7  212.64    1230  213.57
#Mann= 7 ,-1 , 0
       0     .11       0   347.3    .125       0   412.1     .11       0
   455.3     .06       0   608.5     .11       0   883.5     .11       0
   962.9    .125       0
Bank Sta=455.3,608.5
XS Rating Curve= 0 ,0
Exp/Cntr=0.3,0.1

Type RM Length L Ch R = 1 ,26000   ,500,500,500
BEGIN DESCRIPTION:
STEWART CREEK NORTH 52.0
END DESCRIPTION:
XS GIS Cut Line= 3
      3771267.85     10138211.11      3771211.45     10137387.24
      3771017.86     10136911.09
#Sta/Elev= 30
  4174.2  215.56  4248.4  215.41  4354.7   211.8  4396.8   211.6  4424.8  208.11
  4434.8  208.43  4464.9   206.1  4540.2  203.62  4615.3  202.74  4645.3  204.53
  4845.8   204.4  4865.9  203.53  4966.1  202.15  4969.7   200.5    5039     201
    5071  203.68    5093  205.21  5159.4  205.76  5183.5  202.64    5201  204.41
  5212.9  208.19  5222.6  208.34  5308.9  207.97  5397.6  210.41  5406.1  208.65
  5416.3  208.19  5438.5  209.32  5445.7  212.03  5451.1   211.3    5514  214.87
#Mann= 3 , 0 , 0
  4174.2     .11       0  4865.9     .06       0    5071     .11       0
Bank Sta=4865.9,5071
XS Rating Curve= 0 ,0
Exp/Cntr=0.3,0.1

Type RM Length L Ch R = 1 ,25500   ,500,500,500
BEGIN DESCRIPTION:
STEWART CREEK NORTH 51.0
END DESCRIPTION:
XS GIS Cut Line= 3
      3771317.84     10138211.09      3771696.31     10137268.86
      3771667.85     10136761.05
#Sta/Elev= 30
  3984.6  213.79  4082.8  212.42  4113.9  213.05  4262.9  208.93    4322  209.96
  4329.5  209.75  4346.2  207.12  4351.6  207.81  4361.8  206.86  4370.4  205.43
  4375.8  206.41  4394.1  205.14  4598.9  203.95  4615.1   206.8  4620.5  205.94
  4631.2  206.77  4698.4  206.21  4728.2  204.32  4824.8  205.59  4900.6  202.24
  4902.4   200.5    5118     201    5128  202.53  5218.1  204.66  5228.1  205.69
  5308.3  206.78  5328.3  210.12  5368.4   212.9  5458.5  214.55  5508.6  224.82
#Mann= 3 , 0 , 0
  3984.6     .11       0  4900.6    .015       0    5128     .11       0
#XS Ineff= 2 , 0
       0  4631.2  206.77  5241.8       0  205.84
Permanent Ineff=
       F       F
Bank Sta=4900.6,5128
XS Rating Curve= 0 ,0
Exp/Cntr=0.3,0.1
