--- ROBINSON CREEK.prj (project) ---

Proj Title=ROBINSON CREEK Base Level Engineering
Current Plan=p01
Default Exp/Contr=0.3,0.1
English Units
Geom File=g01
Flow File=f01
Plan File=p01
Y Axis Title=Elevation
X Axis Title(PF)=Main Channel Distance
X Axis Title(XS)=Station
BEGIN DESCRIPTION:
ROBINSON CREEK
END DESCRIPTION:
DSS Export Rating Curves= 0
DSS Export Rating Curve Sorted= 0
DSS Export Volume Flow Curves= 0
DXF OffsetX= 0
DXF OffsetY= 0
DXF ScaleX= 1
DXF ScaleY= 10

--- ROBINSON CREEK.p01 (plan) ---

Plan Title=Multiple Run
Program Version=4.10
Short Identifier=Multiple
Geom File=g01
Flow File=f01
Subcritical Flow
K Sum by GR= 0
Std Step Tol= 0.01
Critical Tol= 0.01
Num of Std Step Trials= 20
Max Error Tol= 0.3
Flow Tol Ratio= 0.001
Split Flow NTrial= 30
Split Flow Tol= 0.02
Split Flow Ratio= 0.02
Log Output Level= 0
Friction Slope Method= 1
Unsteady Friction Slope Method= 2
Unsteady Bridges Friction Slope Method= 1
Parabolic Critical Depth
Global Vel Dist= 1 , 1 , 1
Global Log Level= 0
CheckData=True
Encroach Param=-1 ,0,0, 0
BEGIN DESCRIPTION:
Multiple Run
END DESCRIPTION:
Computation Interval=1HOUR
Output Interval=1HOUR
Run HTab= 0
Run UNet= 0
Run PostProcess= 0
Run WQNet= 0
UNET Theta= 1
UNET Theta Warmup= 1
UNET ZTol= 0.02
UNET ZSATol= 0.05
UNET MxIter= 20
UNET MaxInSteps= 0
UNET DtIC= 0
UNET DtMin= 0
UNET MaxCRTS= 20
UNET WFStab= 2
UNET SFStab= 1
UNET WFX= 1
UNET SFX= 1
UNET DSS MLevel= 4
UNET DZMax Abort= 100
UNET Convert EG Bridges= 0
UNET Use Existing IB Tables=-1
UNET Froude Reduction=False
UNET Froude Limit= 1
UNET Froude Power= 10
UNET Time Slicing=0,0, 5
UNET Junction Losses=0
Instantaneous Interval=1HOUR
Write IC File= 0
Write IC File at Sim End=0
Echo Input=False
Echo Parameters=False
Echo Output=False
Write Detailed= 0
WQ AD Non Conservative
WQ ULTIMATE=-1
WQ Max Comp Step=1HOUR
WQ Output Interval=15MIN
WQ Output Selected Increments= 0
WQ Output face flow=0
WQ Output face velocity=0
WQ Output face area=0
WQ Output face dispersion=0
WQ Output cell volume=0
WQ Output cell surface area=0
WQ Output cell continuity=0
WQ Output cumulative cell continuity=0
WQ Output face conc=0
WQ Output face dconc_dx=0
WQ Output face courant=0
WQ Output face peclet=0
WQ Output face adv mass=0
WQ Output face disp mass=0
WQ Output cell mass=0
WQ Output cell source sink temp=0
WQ Output cell source sink nsm=0
WQ Output MaxMinRange=-1
WQ Daily Max Min Mean=-1
WQ Daily Range=0
WQ Daily Time=0
WQ Create Restart=0
WQ Fixed Restart=0
WQ System Summary=0
WQ Use Fixed Temperature=0
Sorting and Armoring Iterations= 10
XS Update Threshold= 0.02
Hydraulics Update Threshold= 0.02
Energy Slope Method= 1
Volume Change Method= 0
XS Weighting Method= 0
Number of US Weighted Cross Sections= 1
Number of DS Weighted Cross Sections= 1
Upstream XS Weight=0.25
Main XS Weight=0.5
Downstream XS Weight=0.25
Number of DS XS's Weighted with US Boundary= 1
Upstream Boundary Weight= 1
Weight of XSs Associated with US Boundary= 0
Number of US XS's Weighted with DS Boundary= 1
Downstream Boundary Weight= 0.5
Weight of XSs Associated with DS Boundary= 0.5
Sediment Output Level= 4
Mass or Volume Output= 0
Output Increment Type= 1
Profile and TS Output Increment= 10
XS Output Flag= 0
XS Output Increment= 10
Disregard all LS=0
Disregard all Conn=0
Disregard all Breaches=0
Disregard all Pumps=0

--- ROBINSON CREEK.f01 (steady flow) ---

Flow Title=Multiple
Program Version=4.10
Number of Profiles= 7
Profile Names=10-year,25-year,50-year,1pct_min,100-year,1pct_plu,500-year
River Rch & RM=ROBINSON CREEK,Reach-1         ,68344
     307     400     527     230     696    2102    1244
River Rch & RM=ROBINSON CREEK,Reach-1         ,67552
    1223    1729    2405    1100    3323   10035    6558
River Rch & RM=ROBINSON CREEK,Reach-1         ,61942
    2047    2947    4150    1917    5789   17483   11653
River Rch & RM=ROBINSON CREEK,Reach-1         ,61130
    2047    2947    4150    1917    5789   17483   11653
River Rch & RM=ROBINSON CREEK,Reach-1         ,56828
    2303    3312    4660    2148    6487   19590   13012
River Rch & RM=ROBINSON CREEK,Reach-1         ,48931
    3560    5231    7467    3489   10537   31821   21710
River Rch & RM=ROBINSON CREEK,Reach-1         ,47829
    3232    4671    6592    3043    9190   27753   18485
River Rch & RM=ROBINSON CREEK,Reach-1         ,42357
    3644    5294    7499    3474   10490   31679   21239
River Rch & RM=ROBINSON CREEK,Reach-1         ,42043
    3644    5294    7499    3474   10490   31679   21239
River Rch & RM=ROBINSON CREEK,Reach-1         ,38959
    3664    5304    7493    3461   10451   31562   21036
River Rch & RM=ROBINSON CREEK,Reach-1         ,34743
    3628    5250    7415    3423   10336   31214   20791
River Rch & RM=ROBINSON CREEK,Reach-1         ,31135
    3900    5663    8018    3709   11201   33826   22630
River Rch & RM=ROBINSON CREEK,Reach-1         ,25196
    4242    6168    8738    4044   12214   36886   24701
River Rch & RM=ROBINSON CREEK,Reach-1         ,22205
    4215    6115    8651    3998   12073   36460   24336
River Rch & RM=ROBINSON CREEK,Reach-1         ,17064
    4368    6328    8942    4127   12463   37638   25055
River Rch & RM=ROBINSON CREEK,Reach-1         ,10458
    4335    6257    8818    4058   12254   37006   24491
River Rch & RM=ROBINSON CREEK,Reach-1         ,5940
    4307    6205    8733    4013   12120   36602   24163
Boundary for River Rch & Prof#=ROBINSON CREEK,Reach-1         , 1
Up Type= 0
Dn Type= 3
Dn Slope=0.0003
Boundary for River Rch & Prof#=ROBINSON CREEK,Reach-1         , 2
Up Type= 0
Dn Type= 3
Dn Slope=0.0003
Boundary for River Rch & Prof#=ROBINSON CREEK,Reach-1         , 3
Up Type= 0
Dn Type= 3
Dn Slope=0.0003
Boundary for River Rch & Prof#=ROBINSON CREEK,Reach-1         , 4
Up Type= 0
Dn Type= 3
Dn Slope=0.0003
Boundary for River Rch & Prof#=ROBINSON CREEK,Reach-1         , 5
Up Type= 0
Dn Type= 3
Dn Slope=0.0003
Boundary for River Rch & Prof#=ROBINSON CREEK,Reach-1         , 6
Up Type= 0
Dn Type= 3
Dn Slope=0.0003
Boundary for River Rch & Prof#=ROBINSON CREEK,Reach-1         , 7
Up Type= 0
Dn Type= 3
Dn Slope=0.0003
DSS Import GetInterval= 0
DSS Import GetPeak= 0
DSS Import FillOption= 0

--- ROBINSON CREEK.g01 (geometry) ---

Geom Title=Existing Conditions
Program Version=4.10

River Reach=ROBINSON CREEK  ,Reach-1
Reach XY= 30
      3797731.15     10252990.93      3794288.23     10250176.84
      3794298.23     10249616.84      3793020.87     10248367.58
      3792253.85     10245682.77      3789502.13     10242860.59
      3787018.19     10241339.16      3785885.86     10241523.27
      3784511.04      10239947.6      3785098.31     10237325.06
      3784638.38     10236597.73      3784809.28     10234720.26
      3785108.42     10233886.67      3786407.41     10232941.66
      3786132.68     10230321.36      3784839.39     10229430.43
      3783311.71      10227251.6      3781595.57     10226323.89
      3780679.66     10225085.41      3780691.47     10224189.73
      3778180.54     10222268.97      3777403.12     10220222.52
      3776346.06     10220324.88      3776147.47      10218655.6
      3774250.85     10218334.08      3772822.56     10216325.77
      3770200.26     10214418.89       3769564.9      10213313.6
      3768369.04     10213454.89      3767188.23     10212376.84

Type RM Length L Ch R = 1 ,68344   ,792,792,792
BEGIN DESCRIPTION:
ROBINSON CREEK 118.0
END DESCRIPTION:
XS GIS Cut Line= 3
      3798177.53     10252746.03      3797799.91     10252858.88
      3797198.65     10253199.36
#Sta/Elev= 30
  4497.3  419.83  4538.7  420.24  4580.5   414.5  4604.4  415.07  4670.6  410.13
  4703.7  408.93  4808.3  407.55  4851.9  404.99  4879.8   406.2  4889.9  404.64
  4916.8  405.39  4939.8   404.3    4962  401.73  4967.7  400.44  4974.2  396.68
  4989.3  391.76  4995.5   387.6  5005.2  389.13    5011  392.17  5032.6  396.07
    5151  400.34  5204.1  403.98  5231.8  407.29  5284.5   408.4  5328.5   413.8
  5436.7  416.36  5452.6  419.47  5474.2  421.25  5539.1  424.02  5582.4  427.53
#Mann= 3 , 0 , 0
  4497.3     .11       0  4974.2     .06       0  5032.6     .11       0
Bank Sta=4974.2,5032.6
XS Rating Curve= 0 ,0
Exp/Cntr=0.3,0.1

Type RM Length L Ch R = 1 ,67552   ,853,853,853
BEGIN DESCRIPTION:
Mapping XS 0cb81d05
END DESCRIPTION:
XS GIS Cut Line= 2
      3797627.56     10251842.25      3796825.74     10252846.65
#Sta/Elev= 30
  4368.3  421.46  4409.7   421.3  4486.5  414.13  4537.8  411.11  4566.7  412.51
  4630.7  409.98  4680.3  402.98  4709.2  402.81    4730  399.78  4744.4  400.75
    4794  397.13  4808.4   398.5  4837.3  397.39  4843.7  395.65  4907.7  391.31
  4957.3  389.43  4986.2  385.15  4998.8  377.98  5029.4  384.46  5135.1  389.17
  5213.5  396.17  5235.9  402.59    5292  403.25  5327.2  407.23    5364  408.35
  5399.3   413.9  5463.3  418.17  5519.3  425.87  5591.4  431.41  5653.5  440.04
#Mann= 4 ,-1 , 0
  4368.3    .125       0  4486.5     .11       0  4957.3     .06       0
  5135.1     .11       0
Bank Sta=4957.3,5135.1
XS Rating Curve= 0 ,0
Exp/Cntr=0.3,0.1

Type RM Length L Ch R = 1 ,66699   ,497,497,497
BEGIN DESCRIPTION:
Mapping XS ac07fe4b
END DESCRIPTION:
XS GIS Cut Line= 2
       3796859.4     10251355.72      3796112.72     10252535.48
#Sta/Elev= 30
  4414.1  390.61  4462.8  391.38  4535.7  390.14  4550.6   389.4  4586.1  383.72
  4621.6   384.1  4635.7  381.69  4693.3  380.01    4918  378.11  4963.8  375.06
  4976.7  373.27  4983.2  369.89  5000.2  372.69  5006.1  372.46  5035.8  378.08
  5048.5  380.62  5130.5  384.82    5179  389.32  5251.9  393.71  5288.4  399.53
    5346  403.47  5434.2  412.76  5506.6  416.99  5570.6   420.3  5592.1  423.56
  5622.4  425.42    5680  425.74  5731.7  428.88    5790  428.96  5810.3  426.93
#Mann= 5 ,-1 , 0
  4414.1     .11       0    4918     .06       0  5035.8     .11       0
  5506.6    .125       0    5790     .11       0
Bank Sta=4918,5035.8
XS Rating Curve= 0 ,0
Exp/Cntr=0.3,0.1

Type RM Length L Ch R = 1 ,66202   ,512,512,512
BEGIN DESCRIPTION:
ROBINSON CREEK 117.0
END DESCRIPTION:
XS GIS Cut Line= 3
      3796433.48     10251022.67      3796139.58     10251563.02
      3795739.04      10252270.5
#Sta/Elev= 30
    4365  394.32  4471.1  392.78  4552.8  386.47  4590.8  385.33  4618.4  381.12
  4634.5     376  4640.2  377.35  4647.8  376.37  4662.1  379.37  4716.1  377.31
  4721.9  378.38  4750.2  375.74  4781.8  375.83  4787.5  374.39  4803.6  375.01
  4869.2  371.86  4950.9  372.21  4976.7  362.05  4986.9  361.28  4994.4  362.31
  5010.3  368.89  5023.8   372.1  5053.6  374.17  5140.2  375.67  5252.8  383.56
  5345.6  387.63    5472  390.23  5749.1  391.32  5780.9  396.04  5793.1  401.06
#Mann= 3 , 0 , 0
    4365     .11       0  4950.9     .06       0  5023.8     .11       0
Bank Sta=4950.9,5023.8
XS Rating Curve= 0 ,0
Exp/Cntr=0.3,0.1

Type RM Length L Ch R = 1 ,65690   ,561,561,561
BEGIN DESCRIPTION:
ROBINSON CREEK 116.0
END DESCRIPTION:
XS GIS Cut Line= 3
      3796043.59      10250737.5      3795741.51     10251230.55
      3795595.94     10252207.94
#Sta/Elev= 30
  4314.3  398.78  4356.8  398.57  4372.2  395.26  4400.6  396.65  4436.1  390.54
  4517.9  385.81  4604.3  382.86  4619.8  380.02  4677.8  379.41  4778.4  375.27
  4851.9   368.4  4913.3  368.95  4973.9  367.38  4980.8  365.08  5002.5  354.34
  5014.2  357.64  5019.3  356.51  5024.5  361.28  5034.6  365.58  5088.6  364.85
  5135.7   366.9  5152.9  365.59  5267.1  371.55  5307.6   370.7  5337.9   372.7
  5702.5  378.07    5803  380.81  5836.1  383.47  5853.5   387.9  5880.7  398.24
#Mann= 3 , 0 , 0
  4314.3     .11       0  4980.8     .06       0  5034.6     .11       0
Bank Sta=4980.8,5034.6
XS Rating Curve= 0 ,0
Exp/Cntr=0.3,0.1

Type RM Length L Ch R = 1 ,65129   ,395,395,395
BEGIN DESCRIPTION:
ROBINSON CREEK 115.0
END DESCRIPTION:
XS GIS Cut Line= 3
      3795776.23     10250553.47      3795400.43     10250962.56
       3794814.4     10251872.95
#Sta/Elev= 30
  4295.1  398.59  4334.5  393.73  4370.3  394.13  4433.8  386.56  4490.5  384.47
  4497.3  382.85    4554  379.72  4639.1  370.67  4681.6  371.87  4759.3  366.76
    4837  363.31    4896  362.41  4932.1  360.02  4953.4  361.58  4980.5   361.9
  4995.7  354.59  5001.7  353.75  5005.2  353.75  5010.9  357.34  5026.1     362
  5119.8  360.48  5192.5  362.31  5307.4  368.88  5364.8  367.94  5422.2  370.15
  5494.9  374.86    5713  385.13  5821.7  391.92  5885.3  397.07  5933.3  399.79
#Mann= 7 ,-1 , 0
  4295.1     .11       0    4896     .11       0  4980.5     .06       0
  5026.1     .11       0  5119.8     .11       0    5713     .17       0
  5885.3     .11       0
Bank Sta=4980.5,5026.1
XS Rating Curve= 0 ,0
Exp/Cntr=0.3,0.1

Type RM Length L Ch R = 1 ,64734   ,453,453,453
BEGIN DESCRIPTION:
ROBINSON CREEK 114.0
END DESCRIPTION:
XS GIS Cut Line= 3
      3795623.48     10250279.14      3795187.71     10250720.02
      3794599.36     10251307.31
#Sta/Elev= 30
  4142.3  399.07  4197.2  393.72  4246.6  392.53  4303.2  384.87    4381  384.61
  4529.5  378.01  4543.6  377.24  4564.9  371.34  4593.2  372.54    4678   361.4
  4699.2  360.12  4748.7  360.96  4798.2  359.09  4861.8  359.47  4925.5  359.98
    4975  360.24    4982  358.78  4989.1  357.28  5001.5  351.41    5005  351.41
  5024.5  358.79  5031.5   359.2  5052.8  356.62    5074  356.42  5102.2  362.09
    5180  361.85  5225.6  364.62  5226.1  364.64  5363.9  376.71  5593.5  388.44
#Mann= 10 ,-1 , 0
  4142.3     .11       0  4748.7     .11       0  4861.8     .11       0
  4925.5     .11       0    4982     .06       0  5024.5     .11       0
  5031.5     .11       0    5074     .11       0  5225.6     .15       0
  5226.1     .17       0
#XS Ineff= 1 ,-1
    4670  4734.6  361.32
Permanent Ineff=
       F
Bank Sta=4982,5024.5
XS Rating Curve= 0 ,0
Exp/Cntr=0.3,0.1

Type RM Length L Ch R = 1 ,64281   ,606,606,606
BEGIN DESCRIPTION:
ROBINSON CREEK 113.0
END DESCRIPTION:
XS GIS Cut Line= 3
      3795323.11     10250016.86      3794928.89     10250385.33
      3794305.88     10251097.33
#Sta/Elev= 30
  4217.9  399.22    4260  395.01  4274.2  391.68  4295.2  391.53  4337.7  384.55
  4387.5  380.64  4493.5  375.62  4564.3   369.3  4592.7   368.4  4599.5  369.38
  4656.2  366.01  4712.8  360.02  4754.8  359.42  4811.9  356.52  4875.5  356.53
  4967.6  358.37  4975.2  358.19  4989.4  351.71  4994.3  351.09  4997.8  351.09
  5010.3  358.25  5017.6  357.86  5088.1  357.54  5095.7  358.95  5116.6  358.48
  5130.8  361.06  5159.3  359.23  5180.2  359.76  5216.3  363.19  5703.6  389.36
#Mann= 8 ,-1 , 0
  4217.9     .11       0  4754.8     .11       0  4875.5     .11       0
  4967.6     .09       0  4975.2     .06       0  5010.3     .09       0
  5017.6     .11       0  5088.1     .11       0
#XS Ineff= 4 ,-1
    4785  4967.6  358.37  5038.8    5093  358.34  5095.7    5120  358.95
  5130.8    5195  361.06
Permanent Ineff=
       T       F       F       F
Bank Sta=4975.2,5010.3
XS Rating Curve= 0 ,0
Exp/Cntr=0.3,0.1

Type RM Length L Ch R = 1 ,63675   ,522,522,522
BEGIN DESCRIPTION:
ROBINSON CREEK 112.0
END DESCRIPTION:
XS GIS Cut Line= 3
      3795190.39      10249642.4      3794238.88     10250273.75
      3793991.32     10250422.07
#Sta/Elev= 30
  3963.6  396.58  3992.5  395.78  4058.7   388.4  4109.8  385.95    4209  384.93
  4230.7  378.97  4311.3   375.5  4347.4  371.16  4398.5  367.99  4446.7  369.46
  4548.9  357.14    4621  357.28  4657.1  353.92  4699.2  354.58  4735.3  352.79
  4866.7   353.4  4924.8  354.34  4981.9  355.26    4997  351.51  5001.2  348.24
  5004.7  348.24  5010.7  352.28    5024  354.98  5090.2  363.26  5126.8  363.52
  5132.7  365.66  5148.2  365.18    5191  369.27  5338.8  391.13  5394.1  394.05
#Mann= 7 ,-1 , 0
  3963.6     .11       0    4621      .2       0  4735.3      .2       0
  4866.7      .2       0  4924.8     .11       0  4981.9     .06       0
    5024     .11       0
Bank Sta=4981.9,5024
XS Rating Curve= 0 ,0
Exp/Cntr=0.3,0.1

Type RM Length L Ch R = 1 ,63153   ,377,377,377
BEGIN DESCRIPTION:
ROBINSON CREEK 111.0
END DESCRIPTION:
XS GIS Cut Line= 3
      3795035.88     10249309.55      3794774.36     10249448.24
      3793888.78     10250228.81
#Sta/Elev= 30
  4202.6  392.92  4290.9  386.82  4326.9   388.5  4392.9  381.56  4491.5  379.04
  4696.3  362.83  4767.4  358.92  4852.8  356.17  4859.4  357.95  4873.6  358.61
    4923  358.64  4951.4  354.95  4973.2     353  4987.2  352.31    4999  345.54
  5002.6  345.54    5015  351.14  5022.6  352.86  5029.2  352.69  5128.8  349.28
  5178.2  350.88  5213.8  349.81  5249.3   352.8  5284.4  353.73  5333.8  352.22
  5390.7  354.97  5440.4  360.99  5532.9  369.31  5596.5  377.01  5679.1   389.4
#Mann= 7 ,-1 , 0
  4202.6     .11       0  4951.4     .11       0  4973.2     .11       0
  4987.2     .06       0  5022.6     .11       0  5029.2     .25       0
  5249.3     .11       0
#XS Ineff= 2 ,-1
  5284.4    5380  353.73
Permanent Ineff=
       F       F
Bank Sta=4987.2,5022.6
XS Rating Curve= 0 ,0
Exp/Cntr=0.3,0.1

Type RM Length L Ch R = 1 ,62776   ,278,278,278
BEGIN DESCRIPTION:
ROBINSON CREEK 110.0
END DESCRIPTION:
XS GIS Cut Line= 3
      3794796.17     10249057.94      3794453.41     10249131.25
      3793732.56     10250111.53
#Sta/Elev= 30
    4184  396.17  4220.5   394.6  4269.9  386.82  4319.4  384.75  4376.6  376.99
  4489.1   368.8  4596.4  365.66  4659.1  359.26  4753.2  365.22  4874.3  352.76
  4918.3  347.86  4974.6  349.87  4981.1  349.28  4993.7  343.57  5003.9  344.62
  5018.4  350.08  5024.8  350.15  5131.3  345.88    5240  349.43  5260.9  352.41
    5311  348.54  5331.9   347.4  5390.4  350.77  5461.4   358.5  5476.1  358.76
  5482.3  356.42  5511.6  361.86  5553.3  361.65  5614.9  367.93  5751.3  385.97
#Mann= 9 ,-1 , 0
    4184     .11       0  4874.3      .2       0  4974.6     .11       0
  4981.1     .06       0  5018.4     .11       0  5024.8     .25       0
    5240     .11       0    5311     .11       0  5614.9     .17       0
#XS Ineff= 3 ,-1
    4880  4974.6  349.87  5260.9    5410  352.41
Permanent Ineff=
       F       F       F
Bank Sta=4981.1,5018.4
XS Rating Curve= 0 ,0
Exp/Cntr=0.3,0.1

Type RM Length L Ch R = 1 ,62498   ,350,350,350
XS GIS Cut Line= 5
       3795045.6      10248885.9      3794204.45     10248990.06
      3794204.45     10248990.06      3793636.74     10249846.83
      3793691.43     10250096.83
#Sta/Elev= 30
       0  399.21   242.7   383.7   283.8  384.18   317.3  377.93   510.4  366.24
   605.1  362.81   647.7  364.82   699.8     361   815.8  357.15  1089.8  351.03
  1148.4  353.95    1177  349.51  1249.2  346.95  1336.4  347.97  1357.5  342.36
  1372.5  347.48  1378.5  347.35  1393.6  344.75  1414.6   341.9  1423.7  342.02
  1444.7  342.83  1486.8  346.15    1532  344.55  1574.1  346.77  1610.2  350.27
  1652.3  347.31  1733.5   348.7  1951.8  356.21  2176.6  381.98  2202.6  387.11
#Mann= 11 ,-1 , 0
       0     .11       0  1249.2     .11       0  1336.4     .06       0
  1372.5     .11       0  1378.5     .25       0  1393.6     .25       0
  1423.7     .25       0  1444.7     .25       0  1486.8     .25       0
  1574.1     .11       0  1733.5     .11       0
#XS Ineff= 2 ,-1
    1200  1279.3  348.33  1610.2    1820  350.27
Permanent Ineff=
       F       F
Bank Sta=1336.4,1372.5
XS Rating Curve= 0 ,0
Exp/Cntr=0.3,0.1

Type RM Length L Ch R = 1 ,62148   ,206,206,206
BEGIN DESCRIPTION:
ROBINSON CREEK 109.0
END DESCRIPTION:
XS GIS Cut Line= 4
      3794415.11     10248263.05      3793931.19     10248879.34
      3793308.36     10249634.55      3793653.11      10250081.2
#Sta/Elev= 30
  3830.8  385.86  3834.5  387.66    3849  384.29  4012.6   380.2  4027.1  377.01
  4062.3  377.42  4076.8  374.51  4214.9  367.99  4237.6  367.35  4397.6  357.76
  4482.6  357.41  4553.1  352.77  4845.5  349.85  4901.8  347.21  4930.1  341.65
    4938  345.67  4979.6  346.56  4987.5  345.41  4999.7  338.87  5016.2  344.94
  5100.8  344.01  5214.2  344.75  5364.1  346.56  5593.3  347.61    5654  349.35
  5676.7  353.13    5818  354.06  5996.4  365.29  6061.3  373.67  6157.5  384.61
#Mann= 10 ,-1 , 0
  3830.8     .11       0  4214.9     .17       0  4237.6     .11       0
  4979.6     .11       0  4987.5     .06       0  5016.2     .11       0
  5100.8     .12       0  5214.2     .12       0  5364.1     .12       0
  6061.3     .17       0
#XS Ineff= 1 ,-1
    4850  4973.2  347.79
Permanent Ineff=
       F
Bank Sta=4987.5,5016.2
XS Rating Curve= 0 ,0
Exp/Cntr=0.3,0.1

Type RM Length L Ch R = 1 ,61942   ,189,189,189
BEGIN DESCRIPTION:
Mapping XS 69b8d8c0
END DESCRIPTION:
XS GIS Cut Line= 2
      3794221.99     10248265.19      3792215.12     10250590.53
#Sta/Elev= 30
    3961  399.68  3968.6  397.35  3975.2  399.76  3989.4  395.33    3996  397.66
  4003.7   395.4  4024.6  397.32  4032.2  394.88  4067.3  395.08  4081.6  391.02
  4159.5  388.75  4173.7  385.03  4613.6  353.59  4734.3  347.77  4890.1   345.4
  4982.2  343.45    5001   335.4  5031.6  343.67  5074.4  345.21  5230.1  347.04
  5315.7  344.92  5520.8  348.24  5846.7     346  6081.4  350.45  6201.1  344.81
  6364.4  358.04  6612.4  368.84  6754.9  367.65  6847.1  372.97  7032.6  374.99
#Mann= 3 , 0 , 0
    3961     .13       0  4890.1     .07       0  5074.4     .13       0
#XS Ineff= 4 ,-1
    4780  4847.3  346.38  5230.1    5445  347.04  5520.8    5997  348.24
  6081.4    6280  350.45
Permanent Ineff=
       F       F       F       F
Bank Sta=4890.1,5074.4
XS Rating Curve= 0 ,0
Exp/Cntr=0.3,0.1

Type RM Length L Ch R = 1 ,61753   ,623,623,623
BEGIN DESCRIPTION:
ROBINSON CREEK 108.0
END DESCRIPTION:
XS GIS Cut Line= 3
      3793808.91     10248467.23      3793617.93     10248699.87
      3791933.93     10250571.37
#Sta/Elev= 30
  4415.4  377.29  4524.9  364.47  4710.1  349.74  4844.7  344.08  4887.3  346.21
  4958.3  343.74  4972.5  342.75  4998.4  331.41  5007.6  333.14  5014.4  340.92
  5021.8  344.39    5107  348.18  5163.1  344.05  5524.9  345.89  5531.6  343.74
  5545.8  346.47  5552.5  343.87    5631  344.31  5737.1  351.72  5800.7  347.34
  5914.3  349.33    5992  342.87  6055.5  343.43  6098.1  347.47  6147.5  343.73
  6169.1  349.84  6622.1  367.22  6756.6  369.42    6806  366.78    7234  375.58
#Mann= 3 , 0 , 0
  4415.4     .15       0  4958.3     .07       0  5021.8     .15       0
#XS Ineff= 3 ,-1
    4775  4887.3  346.21  5737.1    6300  351.72    5107    5700  348.18
Permanent Ineff=
       F       F       F
Bank Sta=4958.3,5021.8
XS Rating Curve= 0 ,0
Exp/Cntr=0.3,0.1

Type RM Length L Ch R = 1 ,61130   ,273,273,273
BEGIN DESCRIPTION:
ROBINSON CREEK 107.0
END DESCRIPTION:
XS GIS Cut Line= 3
      3793708.25     10248231.11       3793371.4     10248370.01
       3791183.9     10249123.49
#Sta/Elev= 30
  4352.6  387.46  4444.6  377.47  4536.9  363.51  4612.6  357.57  4652.3  350.86
  4716.2  344.55  4954.6  340.11  4974.6  339.44  4985.8  333.72    5003  330.76
  5009.5  330.76  5011.8  335.09    5017  338.42  5074.2   339.6  5469.4  341.46
  5757.2  346.75  5812.8  345.94  6088.5  353.13  6145.7  361.44    6151  359.52
  6208.1  360.69  6307.2  355.68  6327.7  358.41    6333   357.1  6358.9  361.64
  6529.3  364.59    6688  373.29  6719.7  377.04  6783.2  376.36  7030.6   391.3
#Mann= 3 , 0 , 0
  4352.6     .15       0  4954.6     .07       0  5074.2     .15       0
Bank Sta=4954.6,5074.2
XS Rating Curve= 0 ,0
Exp/Cntr=0.3,0.1

Type RM Length L Ch R = 1 ,60857   ,313,313,313
BEGIN DESCRIPTION:
ROBINSON CREEK 106.0
END DESCRIPTION:
XS GIS Cut Line= 3
       3793642.2     10248165.15      3792017.24      10248321.4
      3790899.23     10248908.18
#Sta/Elev= 30
  4353.1  380.83  4518.2  359.62    4675  342.73  4769.4  339.78  4980.3  338.68
  4987.5  337.08  5000.4  330.75  5007.2  329.69  5013.7  329.69  5020.5   334.9
  5030.6  338.02  5261.6  338.44  5653.4  342.45  5814.2   346.2  5974.9  352.46
  6103.3  353.46  6176.9  358.31  6296.2   362.9  6323.9  361.54  6362.3  362.26
  6422.8  365.78    6527  368.47  6577.2  371.41  6673.8  380.65  6731.6  379.42
    6748   382.8  6753.6  381.38  6792.1  384.66  7035.2     391  7248.2  393.75
#Mann= 3 , 0 , 0
  4353.1     .15       0  4980.3     .07       0  5030.6     .15       0
Bank Sta=4980.3,5030.6
XS Rating Curve= 0 ,0
Exp/Cntr=0.3,0.1

Type RM Length L Ch R = 1 ,60544   ,670,670,670
BEGIN DESCRIPTION:
ROBINSON CREEK 105.0
END DESCRIPTION:
XS GIS Cut Line= 3
      3793857.51     10247786.68      3793440.85     10247765.84
      3791031.97     10248571.12
#Sta/Elev= 30
  4042.7  393.92  4112.4  383.46  4202.6  373.99  4212.6  371.15  4256.4   371.7
  4272.6  368.93  4458.9  351.43  4553.9  345.04  4648.7  340.46  4737.2  338.35
  4964.6  337.71  4979.7  334.22  4990.2  329.05  4998.2  327.31  5004.7  327.31
  5027.7  336.46    5043  337.41  5154.1  336.41  5496.3  338.65  5665.1  342.14
  6033.2  356.71  6133.3  357.17    6245  362.85  6291.2  362.69  6412.3  369.44
  6575.5  373.69  6670.2  377.89  6719.5  383.16  6877.6  387.76  6999.8  389.11
#Mann= 3 , 0 , 0
  4042.7     .15       0  4964.6     .07       0    5043     .15       0
Bank Sta=4964.6,5043
XS Rating Curve= 0 ,0
Exp/Cntr=0.3,0.1

Type RM Length L Ch R = 1 ,59874   ,526,526,526
BEGIN DESCRIPTION:
ROBINSON CREEK 104.0
END DESCRIPTION:
XS GIS Cut Line= 3
      3794024.19     10246883.89      3793253.35     10247255.43
      3791184.67     10247866.31
#Sta/Elev= 30
  3794.9  377.81  3803.7  377.21  3843.4  383.63  3857.4  382.91  3888.6  376.15
  3916.8  374.64  3933.9  377.49  3956.5  376.61  3979.1  375.06  4007.3  369.45
  4029.9  370.04  4171.1  360.47  4442.5  348.52  4600.8  343.51  4650.6  338.23
  4685.3  341.02  4939.2  334.06  4948.3  333.79    4969  325.78  5021.3  334.47
  5426.2  333.58  5761.6  337.46  6251.7  355.99  6376.8  357.37  6454.3   363.8
    6481  362.93  6559.4  368.22  6664.5  370.54  6741.7  377.45  6807.6  380.59
#Mann= 3 , 0 , 0
  3794.9     .15       0  4939.2     .07       0  5021.3     .15       0
Bank Sta=4939.2,5021.3
XS Rating Curve= 0 ,0
Exp/Cntr=0.3,0.1

Type RM Length L Ch R = 1 ,59348   ,412,412,412
BEGIN DESCRIPTION:
ROBINSON CREEK 103.0
END DESCRIPTION:
XS GIS Cut Line= 3
      3793683.92     10246672.09      3793145.71     10246807.51
      3791176.94     10247724.19
#Sta/Elev= 30
  4040.1  377.79    4067  372.38  4095.1  371.68  4149.5  364.58  4211.3  361.86
    4232   358.8  4259.5  357.14  4324.8   357.9  4355.7   353.7  4465.1  348.16
  4617.8  343.07  4669.9  339.16  4943.6  332.11    4972  330.15  4985.9  322.24
  5000.9  323.77  5011.9  327.17  5017.8  330.89    5034  332.54  5371.9  330.36
  5657.5  334.93    5749  339.41  6017.2  344.74  6154.4  350.17  6348.5  353.87
    6440  358.78  6485.7  362.94  6656.9  371.36  6697.1   371.3  6766.8  376.68
#Mann= 3 , 0 , 0
  4040.1     .13       0  4943.6     .06       0    5034     .13       0
Bank Sta=4943.6,5034
XS Rating Curve= 0 ,0
Exp/Cntr=0.3,0.1

Type RM Length L Ch R = 1 ,58936   ,635,635,635
BEGIN DESCRIPTION:
ROBINSON CREEK 102.0
END DESCRIPTION:
XS GIS Cut Line= 3
      3793735.98     10246401.26      3793114.46     10246429.04
      3791141.24     10247372.69
#Sta/Elev= 30
  4013.7  373.59  4051.9  369.47  4111.9  366.84    4152  369.16  4341.3   357.8
  4392.2   356.4  4532.4  348.43  4665.3  339.91  4964.6  332.96  4978.9  330.07
  4986.8  322.82  4992.6  320.32  4999.6  320.32    5009  325.19  5018.8  327.21
  5041.4  324.85  5053.3  328.12  5069.6  329.32    5115  328.27  5143.2  330.91
  5319.1  329.51  5483.3  329.29  5511.5     328  5551.3  330.17  5738.3  332.62
  6028.8  344.75  6350.2  355.06  6412.4  355.15  6463.3  357.82  6823.1  367.92
#Mann= 4 ,-1 , 0
  4013.7     .11       0  4978.9     .06       0  5069.6     .11       0
  5319.1     .11       0
Bank Sta=4978.9,5069.6
XS Rating Curve= 0 ,0
Exp/Cntr=0.3,0.1

Type RM Length L Ch R = 1 ,58301   ,437,437,437
BEGIN DESCRIPTION:
ROBINSON CREEK 101.0
END DESCRIPTION:
XS GIS Cut Line= 3
      3793364.46     10245331.82      3793277.65     10245623.48
      3790847.07     10247293.64
#Sta/Elev= 30
  3694.2  368.57  3737.6  366.71  3797.8     360  3842.4  360.79  4003.7   350.1
  4171.2   344.1  4254.2     339  4284.5  337.23  4290.6  335.22  4313.7  336.35
  4320.4  334.26    4386  335.53  4586.3  334.03  4846.1  329.51  4968.6  329.34
  4974.6  329.09  4989.5  324.53  5000.9  318.11    5008  318.11  5017.5  325.14
  5031.4  329.21  5255.4  328.28  5377.9  326.12  5470.6  328.51    5593  330.87
    5838  341.46  6255.1   351.4  6312.9  350.05  6384.7  354.57  6947.6  365.74
#Mann= 9 ,-1 , 0
  3694.2     .11       0  4171.2     .15       0  4254.2     .11       0
  4846.1     .11       0  4968.6     .09       0  4974.6     .06       0
  5031.4     .11       0  5255.4     .11       0  5470.6     .11       0
Bank Sta=4974.6,5031.4
XS Rating Curve= 0 ,0
Exp/Cntr=0.3,0.1

Type RM Length L Ch R = 1 ,57864   ,529,529,529
BEGIN DESCRIPTION:
ROBINSON CREEK 100.0
END DESCRIPTION:
XS GIS Cut Line= 3
      3792833.21      10245321.4      3792261.23     10245808.37
      3790705.77      10247146.9
#Sta/Elev= 30
  4248.8  360.79    4302  353.58  4535.1  337.54  4663.3   329.5  4799.7  327.73
  4847.1  327.26    4940   326.1  4976.3  321.87  4982.9  323.58  4990.6  321.94
  4996.2  317.11  5011.4  319.41  5025.7  326.68    5210  324.99  5267.1  326.24
  5308.8  326.33  5337.3  321.82  5359.2  325.42  5387.1  326.32  5571.8   327.7
    5706  330.92  5912.3   339.6  6125.1  343.59  6174.5  341.66  6238.1  346.51
  6287.5  347.76  6323.7  346.95  6514.6  352.03  6819.7  354.48  7052.1  359.18
#Mann= 8 ,-1 , 0
  4248.8     .17       0  4535.1     .11       0  4799.7     .15       0
  4847.1     .11       0    4940     .06       0  5025.7     .11       0
  5267.1     .11       0  5571.8     .11       0
Bank Sta=4940,5025.7
XS Rating Curve= 0 ,0
Exp/Cntr=0.3,0.1

Type RM Length L Ch R = 1 ,57335   ,507,507,507
BEGIN DESCRIPTION:
ROBINSON CREEK 99.0
END DESCRIPTION:
XS GIS Cut Line= 4
      3792725.54     10245040.16      3792382.69     10245227.51
      3790585.81     10246229.39      3790143.09     10246164.28
#Sta/Elev= 30
  4107.4  366.48  4164.4  359.64  4186.3  351.86  4208.1  349.17    4246  351.75
  4449.5  333.67  4652.5  324.59  4848.5  323.29  4938.7  323.05  4961.6  323.81
  4983.4  321.47  5000.7     315  5009.6     315  5010.8  319.66  5018.9  321.77
  5032.5  318.35  5048.5  323.83  5086.2     323    5276   323.7  5687.4  327.63
  5820.3  326.41  5958.3  332.59  5980.6  330.21  6191.1  332.28  6248.3  332.64
  6292.9  333.13  6564.3  337.37  6639.3  341.04  6738.6  346.45  7002.9  359.58
#Mann= 14 ,-1 , 0
  4107.4     .17       0  4449.5     .11       0  4848.5     .11       0
  4938.7     .11       0  4961.6     .06       0  5048.5     .11       0
  5086.2     .11       0    5276     .11       0  6191.1     .15       0
  6248.3     .11       0  6292.9     .15       0  6564.3     .17       0
  6639.3     .11       0  6738.6     .17       0
#XS Ineff= 1 ,-1
  5362.8    5540  325.77
Permanent Ineff=
       F
Bank Sta=4961.6,5048.5
XS Rating Curve= 0 ,0
Exp/Cntr=0.3,0.1

Type RM Length L Ch R = 1 ,56828   ,446,446,446
BEGIN DESCRIPTION:
ROBINSON CREEK 98.0
END DESCRIPTION:
XS GIS Cut Line= 4
      3792697.79      10244547.1      3792326.27     10244599.18
      3790593.63     10245911.68      3790274.19     10245949.87
#Sta/Elev= 30
  3782.8  370.06  4105.9  342.37    4218  335.14  4365.5  325.28  4421.7  323.12
  4744.2  321.28  4885.7  320.23  4964.7  321.72  4979.3   320.6  4993.8  315.02
  4995.6  312.58  5004.6  312.58  5014.6  317.29  5043.8   320.2    5100  319.19
  5129.1  315.61  5143.6  317.14  5172.1  320.72  5357.9  322.82  5528.5  332.59
  5668.5  334.42  5844.2  335.92  5977.9  337.62  6116.3  341.69  6178.7  341.93
  6221.3  343.44  6242.1   341.8  6271.2  344.32  6306.6  343.82  6653.3  357.38
#Mann= 12 ,-1 , 0
  3782.8     .17       0    4218     .11       0  4744.2     .11       0
  4885.7     .11       0  4979.3     .06       0  5043.8     .11       0
  5143.6     .11       0  5668.5     .17       0  5844.2     .11       0
  6116.3     .17       0  6178.7     .15       0  6271.2     .17       0
Bank Sta=4979.3,5043.8
XS Rating Curve= 0 ,0
Exp/Cntr=0.3,0.1

Type RM Length L Ch R = 1 ,56382   ,513,513,513
BEGIN DESCRIPTION:
ROBINSON CREEK 97.0
END DESCRIPTION:
XS GIS Cut Line= 3
       3792107.5     10243734.63       3791871.4     10244366.54
      3790149.22     10245810.96
#Sta/Elev= 30
    3631  360.92    3699  354.51  3936.8  340.63  4203.7  335.55  4305.3   328.6
  4439.5  322.19  4822.1  318.51    4865   319.1  4914.4  317.64  4963.9  318.68
  4971.7  318.14  4995.8  310.93  5004.8  310.93  5021.1  317.75    5028  318.63
  5106.4     317  5142.1  319.22  5177.2  319.39  5532.4   319.8  5624.7  321.27
  5823.8  329.42  5951.3  336.36  5972.1  338.67  6000.7  339.26  6021.6  341.49
  6029.3  340.73  6113.9  347.92  6185.4  351.75  6515.2  360.78  6553.3  362.11
#Mann= 6 ,-1 , 0
    3631     .11       0  4822.1     .11       0  4963.9     .06       0
    5028     .11       0  5177.2     .11       0  6515.2     .17       0
Bank Sta=4963.9,5028
XS Rating Curve= 0 ,0
Exp/Cntr=0.3,0.1

Type RM Length L Ch R = 1 ,55869   ,498,498,498
BEGIN DESCRIPTION:
ROBINSON CREEK 96.0
END DESCRIPTION:
XS GIS Cut Line= 3
       3791801.1     10243573.12      3791020.71     10244435.68
      3789992.01     10245694.53
#Sta/Elev= 30
  3836.8  358.26  3979.4   346.8  4163.3  336.54  4191.7  333.15  4262.6  328.95
  4340.4  325.86  4382.9   325.5  4389.7  326.63  4425.5  324.29  4552.6  322.84
  4651.9   317.3  4708.7  316.27  4888.4  317.44  4963.5  315.24  4984.5  312.36
  4991.9   310.3  4993.9  307.49  5002.9  307.49  5006.5  311.33  5027.3  315.51
  5070.3  314.63    5112  317.07  5190.2  318.24  5389.8  317.29    5575  318.69
  5652.7  321.09  5950.5  341.64  6135.7  351.01  6477.4  356.66  6625.7  356.76
#Mann= 6 ,-1 , 0
  3836.8     .11       0  4651.9     .11       0  4888.4     .11       0
  4963.5     .06       0  5027.3     .11       0  5389.8     .11       0
Bank Sta=4963.5,5027.3
XS Rating Curve= 0 ,0
Exp/Cntr=0.3,0.1

Type RM Length L Ch R = 1 ,55371   ,567,567,567
BEGIN DESCRIPTION:
ROBINSON CREEK 95.0
END DESCRIPTION:
XS GIS Cut Line= 3
       3791631.8      10243373.5      3790690.69     10244095.73
      3789557.18      10244883.9
#Sta/Elev= 30
  3813.7  354.76  4020.8   341.2  4207.6  332.02  4307.3  330.87  4363.5  325.44
  4492.2  325.91  4527.6  332.14  4542.1  329.28  4556.6  329.31  4562.9   327.8
  4670.8  324.91    4785  316.35  4855.7  315.44  4913.7  312.34  4940.9  314.41
  4963.6  314.15  4978.1  310.84  4984.4  307.92    4986  305.54    4996  305.54
  5005.1  310.18  5034.8  314.43  5049.6   315.9  5100.3  315.57  5186.2  311.98
  5258.2  316.12  5681.6  319.55  5759.3  327.15  5896.3  336.95  6380.6   352.8
#Mann= 3 , 0 , 0
  3813.7     .11       0  4963.6     .06       0  5034.8     .11       0
Bank Sta=4963.6,5034.8
XS Rating Curve= 0 ,0
Exp/Cntr=0.3,0.1

Type RM Length L Ch R = 1 ,54804   ,440,440,440
BEGIN DESCRIPTION:
ROBINSON CREEK 94.0
END DESCRIPTION:
XS GIS Cut Line= 3
      3791184.78     10242865.66      3790494.67     10243512.37
      3789357.54     10244705.93
#Sta/Elev= 30
  3742.3  351.92  3906.6   347.2  4168.4  344.14  4557.7  333.27  4614.3  330.29
  4748.6  313.72  4859.2  312.89  4904.3  312.91  4946.7  312.37    4975  309.73
  4981.9  308.42    4984  305.65  5003.3  306.79  5024.4  312.43  5095.2  312.13
  5158.7  308.99  5257.8  313.43    5555  315.56    5767  324.86  5823.6  328.94
  5965.2  329.63  6014.5  333.93  6021.8  332.93  6028.7  334.95  6035.9  333.56
    6057   337.3    6159  343.92    6164  344.15  6262.1   349.7  6336.6  351.65
#Mann= 7 ,-1 , 0
  3742.3     .11       0  4859.2     .15       0  4904.3     .11       0
  4946.7     .06       0  5024.4     .11       0    6159     .17       0
    6164     .11       0
Bank Sta=4946.7,5024.4
XS Rating Curve= 0 ,0
Exp/Cntr=0.3,0.1

Type RM Length L Ch R = 1 ,54364   ,491,491,491
BEGIN DESCRIPTION:
ROBINSON CREEK 93.0
END DESCRIPTION:
XS GIS Cut Line= 3
      3790906.99     10242557.51      3790169.15     10243195.53
      3789075.39     10244584.43
#Sta/Elev= 30
  3624.1  350.35  3924.6  336.53  3959.2  336.53  4001.9  333.72  4008.5  335.72
  4065.6  337.29  4178.6  334.59  4505.4  333.85  4575.6  331.35  4625.8  327.78
  4675.5  321.07  4704.4  320.69  4733.3  316.56  4768.5  315.56  4810.2  310.97
  4842.5  310.65  4888.7  310.76  4924.8  311.18  4967.3  309.11  4981.8   305.6
  4983.2  303.34    5017  306.74  5095.6  310.72  5466.1  313.23  5791.3  333.96
  5945.8  340.24  6016.6  341.15  6043.4  340.35  6191.6  346.48  6367.4  351.22
#Mann= 10 ,-1 , 0
  3624.1     .17       0  3924.6     .11       0  4842.5     .15       0
  4888.7     .11       0  4924.8     .06       0  5095.6     .11       0
  5791.3     .17       0  5945.8     .11       0  6016.6     .17       0
  6191.6     .11       0
Bank Sta=4924.8,5095.6
XS Rating Curve= 0 ,0
Exp/Cntr=0.3,0.1

Type RM Length L Ch R = 1 ,53873   ,524,524,524
BEGIN DESCRIPTION:
ROBINSON CREEK 92.0
END DESCRIPTION:
XS GIS Cut Line= 3
      3790555.44     10242153.86      3789658.57     10243117.33
      3788780.27      10244293.6
#Sta/Elev= 30
  3683.7   345.9    3864  333.29  4042.7  324.54  4196.7  319.35  4422.9  321.36
  4444.4   319.3  4507.9  319.71  4663.6  311.46  4790.8  308.83  4865.3   309.8
  4960.8  309.16  4989.2  305.03  4993.9  302.39  5004.3  302.39  5010.2  305.53
  5017.1  306.33  5074.9  308.85  5104.1  307.97  5145.7  310.23    5159  310.11
  5293.3  310.04  5389.6   311.5  5516.8  310.35  5681.5  313.52  5796.1  320.87
  5825.3  320.99  5846.2  324.85  6017.1  335.56  6152.8  340.05    6468  344.65
#Mann= 8 ,-1 , 0
  3683.7     .17       0  4042.7     .11       0  4865.3     .15       0
  4960.8     .09       0  5074.9     .15       0  5145.7     .11       0
    5159     .15       0  5293.3     .11       0
Bank Sta=4960.8,5074.9
XS Rating Curve= 0 ,0
Exp/Cntr=0.3,0.1

Type RM Length L Ch R = 1 ,53349   ,514,514,514
BEGIN DESCRIPTION:
ROBINSON CREEK 91.0
END DESCRIPTION:
XS GIS Cut Line= 3
      3790364.44     10240890.89      3790164.81     10241359.59
      3788463.42     10244163.41
#Sta/Elev= 30
  2864.4  349.35  3068.9  342.05  3158.1   336.2  3174.5  338.04  3245.2  335.52
  3364.4  332.46  3662.6   325.1  3818.4  322.56  4022.5  321.38    4246   317.8
  4359.4  312.02  4505.9  309.33  4880.4  307.91  4931.3  308.37  4959.4  303.61
  4974.9  306.41    4991  300.89  5038.9  306.81  5083.4  304.89  5118.4  307.65
  5176.9  308.27  5314.1  307.46  5434.3  308.72  5545.8  314.21  5819.4   321.3
  5952.1  324.33    6044  326.96  6155.2   330.7  6466.8  336.79  6653.5  340.39
#Mann= 20 ,-1 , 0
  2864.4     .17       0  3068.9     .15       0  3245.2     .17       0
  3364.4     .11       0  3662.6     .11       0  3818.4     .17       0
  4022.5     .17       0  4359.4     .11       0  4505.9     .11       0
  4880.4     .15       0  4931.3     .09       0  5118.4     .15       0
  5176.9     .11       0  5314.1     .11       0  5545.8     .17       0
  5819.4     .11       0  5952.1     .17       0    6044     .11       0
  6155.2     .17       0  6466.8     .11       0
Bank Sta=4931.3,5118.4
XS Rating Curve= 0 ,0
Exp/Cntr=0.3,0.1

Type RM Length L Ch R = 1 ,52835   ,457,457,457
BEGIN DESCRIPTION:
ROBINSON CREEK 90.0
END DESCRIPTION:
XS GIS Cut Line= 3
      3789490.01     10241149.31      3789117.37     10241968.19
      3788275.43     10244093.73
#Sta/Elev= 30
  3370.3  341.27    3532  331.66  3757.8  327.25  3899.8  319.99  3998.5  311.12
  4124.2  307.43  4358.7  307.04  4595.8  302.61    4610  305.23  4634.3  305.77
  4853.7  306.23  4928.9  306.63    4964  304.51  4999.2  298.19  5009.8  298.19
  5012.6  302.35  5036.8  303.16  5042.3  305.37  5058.3  300.38  5066.7  299.98
  5079.8  305.14  5133.6  307.17  5251.9  307.62  5432.9   314.3  5726.7  321.64
  6032.2  327.95  6112.3  330.98  6381.2   334.7    6435  333.76  6556.2  336.97
#Mann= 10 ,-1 , 0
  3370.3     .11       0  3757.8     .17       0  4124.2     .11       0
  4853.7     .15       0  4928.9     .09       0  5133.6     .15       0
  5251.9     .11       0  5432.9     .17       0  5726.7     .11       0
  6032.2     .17       0
Bank Sta=4928.9,5133.6
XS Rating Curve= 0 ,0
Exp/Cntr=0.3,0.1

Type RM Length L Ch R = 1 ,52378   ,460,460,460
BEGIN DESCRIPTION:
ROBINSON CREEK 89.0
END DESCRIPTION:
XS GIS Cut Line= 3
      3789324.41     10241135.45      3788455.92     10242474.34
        3787692.     10243673.72
#Sta/Elev= 30
  3404.1   341.4  3506.2  331.63  3623.4  326.43  3650.5  322.25  3753.3  322.75
  3944.5  312.24  3997.9  308.95  4174.7  305.62  4208.6  305.17  4395.7  304.36
  4620.2   304.2  4641.3  299.53  4671.6  303.23  4831.3  303.43  4946.5  303.51
  4960.3  301.95  4967.6  297.72  4973.6  297.34  4983.4  290.54    4994  290.54
  4995.1   294.6  5040.3  303.76  5046.2  303.85  5134.2  306.24  5567.6  318.46
  5728.5  318.68  5849.8  313.08  5931.6  319.43  6337.4  333.26    6422  339.01
#Mann= 11 ,-1 , 0
  3404.1     .11       0  3944.5     .17       0  4174.7     .11       0
  4208.6     .15       0  4395.7     .11       0  4831.3     .15       0
  4946.5     .09       0  5040.3     .12       0  5046.2     .15       0
  5134.2     .17       0  6337.4     .11       0
Bank Sta=4946.5,5040.3
XS Rating Curve= 0 ,0
Exp/Cntr=0.3,0.1

Type RM Length L Ch R = 1 ,51918   ,460,460,460
BEGIN DESCRIPTION:
ROBINSON CREEK 88.0
END DESCRIPTION:
XS GIS Cut Line= 3
      3789144.95     10240928.46       3788671.1     10241475.91
      3787296.04     10243356.85
#Sta/Elev= 30
  3486.3  339.49  3677.2  327.76  3755.1  326.97  3797.8  323.93  4039.1   317.3
  4211.4  306.11  4452.1  301.96  4544.3  302.35  4891.7  302.14  4947.2  301.75
    4968  296.02  4997.1  293.33  4998.1  290.22    5009  290.22  5009.5  290.72
  5009.7  293.08  5024.4  300.41  5032.9  298.94  5053.7  301.87  5081.7  303.07
  5158.4  304.38  5200.3  305.59  5384.7  310.79  5399.4  310.84  5440.6  311.87
  5482.3  307.28  5498.5  308.38  5591.2  312.36  5777.3  309.28  6540.3  336.82
#Mann= 12 ,-1 , 0
  3486.3     .11       0  4211.4     .15       0  4544.3     .11       0
  4891.7     .15       0  4947.2     .09       0  5053.7     .15       0
  5081.7     .11       0  5158.4     .17       0  5200.3     .11       0
  5384.7     .17       0  5399.4     .11       0  5498.5     .17       0
Bank Sta=4947.2,5053.7
XS Rating Curve= 0 ,0
Exp/Cntr=0.3,0.1

Type RM Length L Ch R = 1 ,51458   ,644,644,644
BEGIN DESCRIPTION:
ROBINSON CREEK 87.0
END DESCRIPTION:
XS GIS Cut Line= 3
      3788740.12     10240385.53      3787939.59     10241751.96
      3787139.17      10243256.2
#Sta/Elev= 30
  3411.7  331.07  3673.1  318.41    3724  319.01  3980.1  310.41  4236.2  306.56
  4273.3  303.25  4480.9  300.93  4513.7  300.67  4529.4  297.62  4550.9  301.14
  4675.3  300.42    4896  301.16  4967.2  301.28  4982.7  299.06  4992.1  291.32
  4999.3  290.34  5010.5  290.34    5017   297.1  5039.7  299.48  5048.8  300.21
  5070.8   296.1  5098.4  301.54    5113  301.34    5204  301.24    5291  301.94
    5308  301.89  5470.1  308.94  5707.3  312.69  6149.8  315.09  6699.3  335.21
#Mann= 10 ,-1 , 0
  3411.7     .11       0  4480.9     .15       0  4675.3     .11       0
    4896     .15       0  4982.7     .09       0  5039.7     .15       0
    5113     .11       0    5204     .15       0    5291     .11       0
    5308     .17       0
Bank Sta=4982.7,5039.7
XS Rating Curve= 0 ,0
Exp/Cntr=0.3,0.1

Type RM Length L Ch R = 1 ,50814   ,496,496,496
BEGIN DESCRIPTION:
ROBINSON CREEK 86.0
END DESCRIPTION:
XS GIS Cut Line= 3
      3788082.24     10239888.63      3787530.13     10240762.81
       3786982.8     10243195.88
#Sta/Elev= 30
  3172.7  327.73  3652.8  323.05  3808.3  320.01  3923.5  313.66  4133.6  300.01
    4295  298.35  4491.8  297.84  4502.1  293.66  4532.8  298.62  4563.7  294.93
  4594.3  298.45  4733.5  297.97  4887.7  297.85  4946.8  298.33  4963.3  298.67
  4983.8  296.42  4994.1  293.68  4998.7   290.4    5010   290.4  5011.9  293.69
    5017  292.86  5024.8  295.91  5060.3  298.46    5200  298.45  5292.1  298.36
  5513.7  304.57    5697   306.1  5824.3  311.57  6063.8  313.77  6700.5  330.05
#Mann= 10 ,-1 , 0
  3172.7     .11       0  3652.8     .17       0  3923.5     .11       0
    4295     .15       0  4733.5     .11       0  4887.7     .15       0
  4946.8     .11       0  4963.3     .07       0  5060.3     .11       0
    5200     .17       0
Bank Sta=4963.3,5060.3
XS Rating Curve= 0 ,0
Exp/Cntr=0.3,0.1

Type RM Length L Ch R = 1 ,50318   ,403,403,403
BEGIN DESCRIPTION:
ROBINSON CREEK 85.0
END DESCRIPTION:
XS GIS Cut Line= 3
      3787180.47     10239598.86      3787060.86     10240394.75
      3786702.19     10242997.42
#Sta/Elev= 30
  3263.4  328.18    3653  324.47  3963.4  309.41  4175.6  304.96  4316.9  298.76
  4517.4  296.95  4700.5  296.68  4714.2  294.67  4720.7  291.09  4740.8  297.34
  4750.9  297.54  4983.1  296.23  5001.5  289.55  5012.8  289.55  5013.3  290.05
  5013.4  292.18  5023.5   294.8  5063.9  295.39  5319.6  296.67  5336.4  296.88
  5346.5  293.95  5368.5  296.56  5417.2  296.53  5427.3  294.17  5487.3  296.38
  5635.6  301.79  5770.5  307.44  5909.3  307.81  6310.8   324.3  6695.5  329.62
#Mann= 10 ,-1 , 0
  3263.4     .11       0  4517.4     .15       0  4983.1     .09       0
  5063.9     .15       0  5319.6     .17       0  5368.5     .15       0
  5487.3     .11       0  5635.6     .17       0  5909.3     .11       0
  6310.8     .17       0
Bank Sta=4983.1,5063.9
XS Rating Curve= 0 ,0
Exp/Cntr=0.3,0.1

Type RM Length L Ch R = 1 ,49915   ,493,493,493
BEGIN DESCRIPTION:
ROBINSON CREEK 84.0
END DESCRIPTION:
XS GIS Cut Line= 3
      3786738.21     10239498.78      3786582.38     10241426.99
      3786567.23     10242951.62
#Sta/Elev= 30
  3065.5  324.66  3308.6  322.88  3619.6  316.62  3980.8  304.95    4173  303.73
    4253  302.23  4341.9  296.25  4457.7  295.06  4582.7  296.13  4602.8   289.6
  4612.8  288.52  4642.9  295.48  4883.7   295.8  4913.8  293.22  4953.9  295.66
  4991.6  287.42  4993.8  285.16  5005.2  285.16  5024.1  295.64  5064.1  293.32
  5084.1  295.78  5254.1  295.65  5284.1  290.78  5322.6  295.07  5514.1   300.3
  5664.1  308.56  5924.1  314.61    6046  321.02  6151.2  325.05  6524.7  334.44
#Mann= 8 ,-1 , 0
  3065.5     .17       0    4173     .11       0  4457.7     .15       0
  4953.9     .09       0  5024.1     .15       0  5322.6     .17       0
    6046     .11       0  6151.2     .17       0
Bank Sta=4953.9,5024.1
XS Rating Curve= 0 ,0
Exp/Cntr=0.3,0.1

Type RM Length L Ch R = 1 ,49422   ,491,491,491
BEGIN DESCRIPTION:
ROBINSON CREEK 83.0
END DESCRIPTION:
XS GIS Cut Line= 4
      3786688.57     10239460.16      3786066.63     10240918.26
       3786170.1     10242262.12       3786495.3     10242956.61
#Sta/Elev= 30
  2854.6  323.58  3457.2  312.84  3586.1  314.69  3774.3  309.14  4346.9  297.52
  4482.7  293.02  4512.8  286.04  4524.4  285.95  4542.9  294.51  4713.4   294.5
  4803.7   294.1  4883.9  294.45  4974.2  294.68  4984.2  292.97  4998.6   284.3
    5010   284.3  5034.4  294.05  5040.6  294.09  5114.6  294.14  5144.7  294.24
  5164.8  289.44  5184.8  293.63  5296.3  296.57  5505.8  310.74  5649.4  315.46
  5971.3  316.97  6062.9  316.91  6072.5  316.53  6237.9  319.26  6554.5   334.5
#Mann= 15 ,-1 , 0
  2854.6     .17       0  3774.3     .11       0  4346.9     .15       0
  4713.4     .15       0  4803.7     .15       0  4883.9     .15       0
  4974.2     .09       0  5034.4     .12       0  5040.6     .15       0
  5114.6     .15       0  5296.3     .17       0  5649.4     .11       0
  5971.3     .17       0  6062.9     .11       0  6072.5     .17       0
Bank Sta=4974.2,5034.4
XS Rating Curve= 0 ,0
Exp/Cntr=0.3,0.1

Type RM Length L Ch R = 1 ,48931   ,494,494,494
BEGIN DESCRIPTION:
ROBINSON CREEK 82.0
END DESCRIPTION:
XS GIS Cut Line= 3
      3786367.87     10240211.04      3785773.85     10241312.47
      3784667.86     10241911.07
#Sta/Elev= 30
  3748.6  312.72  3856.2  308.96  3924.9  306.94  4050.6  304.31  4464.3  299.19
  4612.1  293.93  4647.9  285.02  4664.1  291.46    4686  293.93  4724.2  289.98
  4833.6  293.35  4921.2  290.07  4975.5  294.76  4981.2  293.23    5000  284.37
  5001.7  278.86  5018.4  278.86  5031.9  289.56  5048.1  292.96    5166  293.86
  5424.8  293.63  5556.1  293.99  5572.2  290.59  5599.8  293.82  5725.4   294.3
  5757.3   289.7  5791.4  293.82  5954.6  295.06  6149.1  312.54  6257.6  318.01
#Mann= 14 ,-1 , 0
  3748.6     .17       0  3856.2     .11       0  3924.9     .17       0
  4050.6     .11       0  4464.3     .15       0  4833.6     .15       0
  4921.2     .13       0  4975.5     .12       0  4981.2     .09       0
  5048.1     .13       0    5166     .15       0  5424.8     .15       0
  5572.2     .15       0  6149.1     .17       0
#XS Ineff= 1 ,-1
    4560  4975.5  294.76
Permanent Ineff=
       F
Bank Sta=4981.2,5048.1
XS Rating Curve= 0 ,0
Exp/Cntr=0.3,0.1

Type RM Length L Ch R = 1 ,48437   ,608,608,608
BEGIN DESCRIPTION:
ROBINSON CREEK 81.0
END DESCRIPTION:
XS GIS Cut Line= 3
      3786017.88     10240061.03      3785425.36     10240973.78
      3784517.85     10241661.07
#Sta/Elev= 30
  3911.8  312.29  4297.4  302.43  4332.6  302.78  4640.2  298.17  4860.6  293.15
  4931.2  292.87  4937.2  291.62  4952.3  288.87  4958.8  280.42  5003.5  282.72
  5024.3  291.97  5117.9  293.01    5147  291.91    5160  287.88  5188.7  291.53
  5217.8  287.95  5267.7  289.59  5282.2  287.29  5303.1  290.89  5332.2  287.35
  5382.1  291.92  5396.7  289.58  5452.9  289.34  5473.7  285.46  5502.8   290.3
  5578.6  292.12  5837.8  294.96  5902.3  298.58  5975.4  306.64  6138.4  318.82
#Mann= 11 ,-1 , 0
  3911.8     .17       0  4297.4     .11       0  4332.6     .17       0
  4640.2     .11       0  4860.6     .15       0  4931.2     .12       0
  4937.2     .09       0  5024.3     .15       0  5188.7     .15       0
  5578.6     .11       0  5975.4     .17       0
#XS Ineff= 1 ,-1
  5117.9    5610  293.01
Permanent Ineff=
       T
Bank Sta=4937.2,5024.3
XS Rating Curve= 0 ,0
Exp/Cntr=0.3,0.1
